HEC-RAS study GRNBRRRV.prj: GRNBRRRV

--- GRNBRRRV.g01 (geometry) --- (continued)

Type RM Length L Ch R = 1 ,300426  ,376.6,403,426.6
XS GIS Cut Line= 3
 2290566.8409302533307.532652185 2289890.2471716532836.659968834
2289794.24400315532635.510473033
#Sta/Elev= 30
       0 2611.28    67.1 2570.04    89.8  2557.9   100.7 2553.15   124.3 2548.88
   151.2 2546.81   256.5  2547.6     359 2549.57   403.3 2552.81   495.5 2547.48
   543.8 2547.55   571.3 2544.17   592.3 2543.57   620.3  2541.7   675.8 2541.66
   690.5  2541.7   697.4 2543.88     705 2549.31   709.9 2555.38   719.1 2569.28
   724.5 2573.96   774.4 2576.99   788.4 2579.64   802.5 2580.23   845.9  2591.6
   868.1 2599.44   933.5 2629.82    1001 2667.81  1009.9 2671.46  1047.2 2694.39
#Mann= 4 ,-1,0
       0      .1       0     570    .025       0   592.3    .035       0
   697.4      .1       0
Bank Sta=592.3,697.4
XS Rating Curve= 0 ,0
Exp/Cntr(USF)=0,0
Exp/Cntr=0.3,0.1

Type RM Length L Ch R = 1 ,300023  ,530.2,526,522.1
XS GIS Cut Line= 2
2290739.95881391533225.1350660142290059.63177271532289.843264512
#Sta/Elev= 30
       0 2666.21    67.6  2643.6      80 2636.76      89  2632.2   117.2 2609.03
   183.2 2566.08   208.8 2552.64   228.9 2545.58   306.6  2545.7   480.9 2549.13
   572.5 2546.08   578.7 2546.13   584.4 2543.69   588.6 2541.46   593.5 2541.03
   727.2 2541.03   738.6 2543.87   752.9 2555.03   770.1 2556.71   775.8 2558.75
   795.8 2574.65   801.2    2577   849.6 2587.66   876.8 2591.75   900.2 2597.53
   979.3 2623.75   999.2 2631.65  1042.1 2650.52  1142.5 2704.09  1156.6 2710.32
#Mann= 6 ,-1,0
       0     .12       0      80      .1       0     540    .025       0
   572.5      .1       0   584.4    .035       0   738.6      .1       0
Bank Sta=584.4,738.6
XS Rating Curve= 0 ,0
Exp/Cntr=0.3,0.1

Type RM Length L Ch R = 1 ,299497  ,495.7,505.7,526.2
XS GIS Cut Line= 2
2291121.26806321532815.1728955922290495.53769266532026.027026214
#Sta/Elev= 30
       0 2679.91      62 2654.71    85.5  2643.9   114.9 2627.65   155.7 2600.58
   201.3 2561.09   227.1 2543.94   246.4  2542.4   329.6 2545.15   354.8 2543.95
   392.3 2545.78   431.4 2544.74     472 2546.78   477.7 2546.04   489.1 2540.81
   492.6 2539.88   640.7 2539.82   648.5 2540.86   677.8 2543.99   727.4 2543.58
   742.1 2551.13   747.9 2552.69   758.1 2553.17   773.4  2551.5   790.9 2554.67
   810.8  2560.3   827.9 2567.91   890.5 2602.46   910.5 2612.28  1007.1 2666.36
#Mann= 5 ,-1,0
       0      .1       0     390     .08       0   489.1    .035       0
   648.5    .025       0     760      .1       0
Bank Sta=489.1,648.5
XS Rating Curve= 0 ,0
Exp/Cntr=0.3,0.1

Type RM Length L Ch R = 1 ,298991  ,414.5,406.7,360.7
XS GIS Cut Line= 3
2291534.62225315532644.8078523162291024.59881485531829.818008189
2290807.35090917531678.674479399
#Sta/Elev= 30
       0 2668.67   100.2 2650.91     163 2634.32   245.9 2595.51   259.8 2586.18
   315.7 2556.86   361.4 2542.29   410.1 2540.92   532.8 2543.78   584.9 2545.25
   596.4 2539.86   602.3 2538.23   745.1 2538.01   749.8 2539.28   782.2 2538.97
   815.9 2537.92   823.4 2539.51   830.1 2543.04   834.5 2543.37   872.5 2542.66
   889.6 2538.71   929.1 2539.82   961.9 2549.43   986.3 2546.62  1010.7 2554.33
  1044.8 2572.39  1132.5 2631.46    1149  2644.8  1169.1 2663.76  1226.1 2708.45
#Mann= 6 ,-1,0
       0      .1       0   532.8     .08       0   596.4    .035       0
   749.8     .08       0   782.2    .035       0   823.4      .1       0
#XS Ineff= 2 , 0
       0                   966.8       0    2556
Permanent Ineff=
       F       F
Bank Sta=596.4,823.4
XS Rating Curve= 0 ,0
Exp/Cntr=0.3,0.1

Type RM Length L Ch R = 1 ,298585  ,337.5,333.4,326.8
XS GIS Cut Line= 2
2291986.90821887532351.7663717282291106.79244218 531427.44768188
#Sta/Elev= 30
       0 2681.39   108.4  2663.7     149 2651.29   196.2 2629.91     346 2547.92
   357.4  2543.2   515.9  2539.5   620.5 2543.72   647.8 2538.04   665.8    2540
   688.8 2537.82   699.5 2536.09   781.3 2537.43   824.3 2539.44   848.6 2537.61
   859.7 2536.08   906.3 2537.41   926.1 2539.06   949.5 2536.66   968.5 2538.55
   982.7 2535.61  1003.3  2536.8  1030.9  2546.9  1050.6 2547.74  1064.7  2551.7
  1104.4 2579.97  1135.1  2604.5  1169.4 2638.57  1224.2 2676.69  1276.3 2707.91
#Mann= 6 ,-1,0
       0      .1       0   620.5     .08       0   688.8    .035       0
   781.3     .08       0   848.6    .035       0   906.3      .1       0
Bank Sta=688.8,906.3
XS Rating Curve= 0 ,0
Exp/Cntr=0.3,0.1

Type RM Length L Ch R = 1 ,298251  ,344.2,358.1,274.9
XS GIS Cut Line= 2
2292282.51311966532104.5349253322291431.85459552531323.760529244
#Sta/Elev= 30
       0 2676.69    34.5 2666.61    75.9 2651.09   171.1 2613.06   258.8 2573.36
   342.1 2542.94   369.2 2539.95   420.2 2539.66   451.3 2539.81   513.7 2537.85
   550.4 2540.35   590.1 2538.77   627.6 2541.56   691.2 2539.15   730.7 2540.64
   738.5 2536.22   744.4 2533.45   817.6 2533.33   842.4 2533.31   893.6 2533.24
   963.7 2533.18  1006.2 2533.11  1023.2 2536.14  1031.7 2540.15  1040.2 2545.88
    1052 2546.73  1057.9 2549.55  1099.9 2590.88  1137.9  2619.4  1154.7 2641.12
#Mann= 12 ,-1,0
       0      .1       0   420.2     .08       0   451.3      .1       0
   590.1     .07       0   691.2     .08       0   738.5    .035       0
   817.6     .08       0   842.4      .1       0   893.6     .08       0
   963.7    .035       0  1023.2     .08       0  1031.7      .1       0
Bank Sta=738.5,1023.2
XS Rating Curve= 0 ,0
Exp/Cntr(USF)=0,0
Exp/Cntr=0.3,0.1

Type RM Length L Ch R = 1 ,297893  ,304.5,291.7,279.8
XS GIS Cut Line= 3
2292521.08307402531841.8669957842291653.55596725531162.304095485
2291508.96811612 531152.66490541
#Sta/Elev= 30
       0 2656.32    72.3 2625.85   128.2 2607.56   173.9  2586.5   234.6  2564.7
   260.4 2558.61   303.2 2554.78   336.5 2541.76   351.6  2538.1   508.3 2540.44
   539.8  2539.8   553.9 2536.62   576.7 2538.26   736.2 2537.09     786 2538.59
   819.2 2536.17   844.6 2537.24   904.3 2532.58  1002.1 2531.24  1009.7 2532.59
  1038.3 2537.36  1068.2 2537.42  1088.5 2545.64  1107.4  2545.3  1111.4 2547.18
  1132.3 2568.81  1159.5  2593.3    1179 2608.54  1222.5 2638.52  1246.9  2648.4
#Mann= 5 ,-1,0
       0      .1       0     540     .08       0     860      .1       0
   904.3    .035       0  1009.7      .1       0
Bank Sta=904.3,1009.7
XS Rating Curve= 0 ,0
Exp/Cntr(USF)=0,0
Exp/Cntr=0.3,0.1

Type RM Length L Ch R = 1 ,297601  ,542.6,493.8,464.9
XS GIS Cut Line= 3
2292736.81176827531448.4383469162291747.96378113 530908.63068188
2291504.90653301530980.637710677
#Sta/Elev= 30
       0 2631.82    64.5 2611.72   110.1  2592.8   135.5 2584.27     224 2541.61
   233.1 2539.94     336  2539.8   374.3 2538.03   388.1 2535.47   433.7 2535.07
   716.2 2538.12   852.9 2537.55   866.7 2536.05  877.93 2532.82   889.4 2530.59
   980.5 2530.59  1005.2 2532.71  1016.9 2534.47    1070 2535.06  1108.8 2534.91
  1130.5  2532.6  1171.9 2534.34  1205.6  2532.1  1209.8 2532.82  1230.7 2544.13
  1255.7 2542.37  1305.8 2569.34  1314.1 2574.71    1335 2592.21  1380.1 2618.65
#Mann= 5 ,-1,0
       0      .1       0     310     .08       0     650      .1       0
  877.93    .035       0  1005.2      .1       0
#XS Ineff= 2 , 0
                         1231.21         2553.47
Permanent Ineff=
       F       F
Bank Sta=877.93,1005.2
XS Rating Curve= 0 ,0
Exp/Cntr=0.3,0.1

Type RM Length L Ch R = 1 ,297108  ,562.2,411.2,293.8
XS GIS Cut Line= 3
2292970.89773105530588.7277727072291964.41984718530542.986133156
2291452.42680992530925.918041203
#Sta/Elev= 30
       0 2603.03   105.6 2581.17   182.2 2570.37     267 2568.81     299 2557.54
   335.1  2552.4   363.1 2541.69   491.2 2536.53   615.8 2537.11   639.4 2533.83
   707.5 2533.92   775.8 2530.35   909.4  2530.4   995.7 2532.59  1111.4  2529.8
  1143.6 2534.61  1218.2 2530.66    1315 2529.38  1402.4 2533.36  1422.4 2529.16
  1442.4 2537.94  1465.3 2540.18  1475.1 2543.55  1487.3 2543.68  1503.6 2539.62
  1529.4 2541.41  1572.3 2558.71  1592.2 2571.21  1603.7 2583.89  1646.9 2604.77
#Mann= 4 ,-1,0
       0      .1       0   775.8    .035       0   909.4     .08       0
    1000      .1       0
#XS Ineff= 2 , 0
                         1472.45         2554.42
Permanent Ineff=
       F       F
Bank Sta=775.8,909.4
XS Rating Curve= 0 ,0
Exp/Cntr=0.3,0.1

Type RM Length L Ch R = 1 ,296696  ,507.1,505.5,504.6
XS GIS Cut Line= 3
2291949.96106206 529798.358699852291887.30632657530477.921600149
2291451.13297567530882.767583305
#Sta/Elev= 30
       0 2740.68      43 2729.03    95.2 2708.79   119.3 2696.13   163.5 2667.86
   219.7 2625.44   308.1 2579.93   328.2 2567.58   360.3 2539.91   383.1 2529.85
     525 2529.86   569.2 2532.94   593.3 2529.28   692.2 2532.99   768.6 2527.69
   816.6 2527.86   842.6 2533.27   876.6 2533.17   904.8 2528.92   919.1 2533.27
   958.7 2529.21  1054.9 2532.36  1071.9 2529.56  1100.2 2538.82  1134.2  2543.5
  1161.5 2538.76  1192.9 2539.48  1210.6 2543.32  1232.5 2553.19  1277.5 2580.32
#Mann= 6 ,-1,0
       0      .1       0     340    .025       0   383.1    .035       0
     525      .1       0     640     .08       0  702.45      .1       0
#XS Ineff= 2 , 0
                         1134.99          2562.5
Permanent Ineff=
       F       F
Bank Sta=383.1,525
XS Rating Curve= 0 ,0
Exp/Cntr(USF)=0,0
Exp/Cntr=0.3,0.1

Type RM Length L Ch R = 1 ,296191  ,605.9,603,602
XS GIS Cut Line= 2
2291442.12388835529751.6912024812291351.02430571530865.936789097
#Sta/Elev= 30
       0 2767.86    37.6 2762.31    53.7 2754.97     162 2678.16   174.1 2665.27
   182.1 2649.53   187.4 2643.62   226.2 2623.63   246.3 2618.01   281.4 2596.83
   318.6 2578.18   354.7 2554.86   390.8 2540.08   410.3 2527.64   414.9 2525.44
   523.2 2525.41   535.3 2527.92   571.4 2531.87   627.6 2529.42     756 2531.04
   784.1 2526.67   856.5 2530.56   904.5 2528.02   924.6 2540.57   932.6 2542.37
   972.7 2535.21  1008.8 2537.88  1032.9 2544.65  1093.1 2576.74    1118 2585.62
#Mann= 4 ,-1,0
       0      .1       0   410.3    .035       0   535.3    .025       0
     580      .1       0
#XS Ineff= 2 , 0
                          933.63         2570.48
Permanent Ineff=
       F       F
Bank Sta=410.3,535.3
XS Rating Curve= 0 ,0
Exp/Cntr=0.3,0.1

Type RM Length L Ch R = 1 ,295588  ,499.9,503.5,504.2
XS GIS Cut Line= 2
2290821.11920248529817.0855081952290767.07101241530865.769764285
#Sta/Elev= 30
       0 2693.89    32.1 2690.01    56.2  2685.3    92.2 2675.03   119.1 2662.81
   163.8 2639.31   188.3 2621.18   216.4 2593.91   224.4 2584.06   244.8 2567.44
  283.47 2523.97   288.5 2522.22   393.3 2522.69   416.6  2521.5   448.7 2527.29
     489 2526.02   508.8 2527.16   532.8 2530.96   564.8 2531.75   580.9 2533.91
   644.9  2535.6     693 2534.13     709 2536.49   729.1 2535.03   797.1 2534.19
   865.6 2535.75   901.3 2539.22   957.7 2547.97   977.4  2549.3  1050.1 2569.38
#Mann= 4 ,-1,0
       0      .1       0     220     .12       0  283.47    .035       0
   393.3      .1       0
#XS Ineff= 2 , 0
                          707.15         2552.56
Permanent Ineff=
       F       F
Bank Sta=283.47,393.3
XS Rating Curve= 0 ,0
Exp/Cntr=0.3,0.1

Type RM Length L Ch R = 1 ,295084  ,428.4,466.3,483.2
BEGIN DESCRIPTION:
c/e of 0.5/0.7 used to correct drawdown
END DESCRIPTION:
XS GIS Cut Line= 3
2290393.64112805529891.5735990222290304.06935673530061.026629398
2290271.33280993530757.191243684
#Sta/Elev= 30
       0 2634.02      29 2627.83    60.6 2616.93   119.5  2585.9   151.1 2566.25
   173.7 2549.21   191.7 2533.86   191.7 2533.82   199.8 2529.37   206.22522.078
   207.8 2520.83   211.8  2520.5     336 2520.53   343.2 2522.14     352 2525.47
   363.8 2527.03   408.1 2528.24   460.1 2531.73   504.2 2530.08   524.5 2535.51
   532.2 2534.93   544.2 2530.82   552.2 2531.93   568.2 2530.69     666 2531.92
   708.4 2538.73   740.4 2550.88   771.8  2558.2   800.5 2562.08   888.6 2570.53
#Mann= 5 ,-1,0
       0      .1       0   191.7     .12       0   206.2    .035       0
   343.2    .025       0   363.8      .1       0
#XS Ineff= 2 , 0
                          523.38         2551.96
Permanent Ineff=
       F       F
Bank Sta=206.2,343.2
XS Rating Curve= 0 ,0
Exp/Cntr=0.7,0.5

Type RM Length L Ch R = 1 ,294618  ,221,338.3,390
XS GIS Cut Line= 3
2290185.98927831529788.7195097752289884.76458846529988.732703834
2289735.35714229530473.102005111
#Sta/Elev= 30
       0 2597.05      94 2575.61   145.9 2561.54   210.5 2541.27   223.8 2536.07
   237.5 2529.18   246.9 2526.79   261.2 2527.47   290.1  2526.1   319.1 2526.09
   328.7 2522.15   333.5 2521.16   343.1 2520.81   363.6 2523.51   381.6 2521.86
   399.7 2519.32   567.2 2519.28   575.5 2519.66   583.9 2522.02   588.1 2524.35
   600.6 2526.65   613.2 2532.25   646.7 2535.28   663.1 2547.84   667.6  2550.1
   705.3 2559.88   713.7  2560.8   751.3 2568.16   801.6 2582.43   868.5 2599.59
#Mann= 4 ,-1,0
       0      .1       0     340     .08       0   381.6    .035       0
   583.9      .1       0
Bank Sta=381.6,583.9
XS Rating Curve= 0 ,0
Exp/Cntr(USF)=0,0
Exp/Cntr=0.3,0.1

Type RM Length L Ch R = 1 ,294280  ,182.7,229.4,264.9
XS GIS Cut Line= 3
2290184.08455999529738.4471483412289742.30936447 529867.35039236
2289252.97763232530122.653904786
#Sta/Elev= 30
       0 2598.36   138.3 2565.01   191.6 2550.22   212.4 2542.99   250.5 2534.52
   308.2 2527.76   366.6 2526.44   373.1 2525.21   383.3 2520.79     390  2519.9
   467.1 2524.05   489.8 2524.09   516.5 2523.23   530.3 2520.12   540.2 2517.73
   645.7 2517.62   661.1 2517.95   664.7 2520.12   680.3 2530.11   692.7 2532.81
   710.7 2533.38   715.3 2534.98   719.8 2538.23   728.8 2547.75   751.4 2577.32
   759.6 2583.92   864.1 2626.71   936.3 2658.14   945.4 2660.99  1012.1 2691.54
#Mann= 5 ,-1,0
       0      .1       0   500.2     .08       0   530.3    .035       0
   664.7     .08       0   720.2      .1       0
Bank Sta=530.3,664.7
XS Rating Curve= 0 ,0
Exp/Cntr(USF)=0,0
Exp/Cntr=0.3,0.1

Type RM Length L Ch R = 1 ,294050  ,424,445.4,470.5
XS GIS Cut Line= 3
2290184.55143432529687.0292906142289773.59655962529723.429294669
2289176.28411794529692.327609023
#Sta/Elev= 30
       0 2599.85   136.9 2566.89   221.2  2542.8   253.4 2535.68   293.8 2530.98
   329.7 2531.56     426 2525.72     434  2524.3     442 2520.54   454.1 2518.68
   510.1 2520.55   534.1 2519.25   562.2 2520.37   582.2 2517.03   638.3 2516.89
   650.3 2517.05   655.9 2519.93   674.3 2529.97   690.4 2533.09   694.4 2535.55
   710.4 2549.02   718.4 2560.15   754.4 2596.53   766.3 2605.71   814.5 2630.47
   822.5 2635.89   850.6 2659.48   866.6 2670.12   950.7 2719.27  1010.7 2757.26
#Mann= 4 ,-1,0
       0      .1       0   562.2    .035       0   655.9     .08       0
  672.56      .1       0
#XS Ineff= 2 , 0
          338.73 2549.76
Permanent Ineff=
       F       F
Bank Sta=562.2,655.9
XS Rating Curve= 0 ,0
Exp/Cntr(USF)=0,0
Exp/Cntr=0.3,0.1

Type RM Length L Ch R = 1 ,293605  ,488.6,515.8,540.6
XS GIS Cut Line= 2
2290176.94111564529487.291735489     2289243.487      529103.548
#Sta/Elev= 30
       0 2582.24   173.8 2542.42   216.7 2536.14   273.3 2529.66   394.4 2526.72
   463.6 2519.84   489.5 2520.12   506.8 2516.59   523.2 2513.92   587.6 2513.86
     602 2514.17   607.1 2516.38   627.9 2521.69   649.6 2532.84   653.9 2536.99
   670.3 2574.07   675.5 2583.16   684.1 2593.04     701  2607.9   716.3 2624.15
   756.2 2652.34   787.9 2678.96   800.9 2686.88   861.5  2736.7   874.4 2745.35
     935 2794.49   949.2 2807.95   979.9 2833.59   991.2 2847.56  1009.3  2865.2
#Mann= 3 ,0,0
       0      .1       0   506.8    .035       0   607.1      .1       0
Bank Sta=506.8,607.1
XS Rating Curve= 0 ,0
Exp/Cntr=0.3,0.1

Type RM Length L Ch R = 1 ,293089  ,490,505.4,517.9
XS GIS Cut Line= 2
2290380.68588835529269.559685864     2289615.121      528529.195
#Sta/Elev= 30
       0 2582.38    28.5  2574.5   121.4 2553.98     248 2532.33     317  2527.5
   390.2 2526.23   467.4 2521.98   534.9 2513.01   554.62512.157   564.4 2511.16
   639.9 2511.26   648.4 2512.68   662.9 2517.56   673.8 2525.96   685.1 2538.03
   713.5 2558.26   758.8  2583.5   771.6 2589.28     821 2619.63   922.8 2690.16
   976.6 2737.31   990.2 2746.12    1002 2756.74  1013.5    2765    1019 2774.19
  1024.7 2786.51  1027.5 2789.98  1047.3 2803.79    1058 2818.94    1065  2826.8
#Mann= 4 ,-1,0
       0      .1       0     520    .025       0   554.6    .035       0
   648.4      .1       0
Bank Sta=554.6,648.4
XS Rating Curve= 0 ,0
Exp/Cntr=0.3,0.1

Type RM Length L Ch R = 1 ,292584  ,501.3,501.7,504.4
XS GIS Cut Line= 2
2290671.80392556529017.248103233     2290089.561      528169.574
#Sta/Elev= 30
       0  2605.9    65.9 2580.76   116.5 2563.75   201.2 2547.16   252.9 2534.34
   296.1 2525.91   446.5 2521.24   472.7  2519.2   506.1  2511.9   514.7  2510.5
   615.4 2510.51   630.9 2511.95   647.1 2514.08   672.9 2525.85     694 2551.37
   713.4  2567.1     727 2584.05     742 2595.11   757.1 2610.71   783.6 2630.87
   829.9 2670.17   839.8 2676.38   868.6 2699.49     939  2759.7   954.9 2774.58
   972.1 2798.29   986.5  2812.7  1002.6  2844.4  1006.6 2850.64  1028.4 2868.36
#Mann= 4 ,-1,0
       0      .1       0     480    .025       0   506.1    .035       0
   630.9      .1       0
Bank Sta=506.1,630.9
XS Rating Curve= 0 ,0
Exp/Cntr=0.3,0.1

Type RM Length L Ch R = 1 ,292082  ,497.6,498.1,491.4
XS GIS Cut Line= 2
     2291030.412      528656.114     2290516.593       527904.99
#Sta/Elev= 30
       0 2595.24    55.5 2572.38     115 2545.74   144.7 2534.39   167.8 2527.31
   195.2 2524.19   236.8 2522.26   366.3 2520.99   372.1 2519.98   391.3 2512.39
   396.1 2510.33   400.9 2509.75   576.4 2509.78   580.3 2509.97   587.9 2512.93
   594.8 2516.56   604.5 2519.22   625.3 2521.71   638.4 2520.98   642.6 2522.01
   691.7 2555.68   720.8 2572.37   737.6 2579.56   769.1 2596.65   776.2 2599.71
   808.1 2620.05   823.9 2629.03   846.4 2638.82   855.5  2645.2   910.1 2660.21
#Mann= 3 ,-1,0
       0      .1       0   391.3    .035       0   587.9      .1       0
Bank Sta=391.3,587.9
XS Rating Curve= 0 ,0
Exp/Cntr=0.3,0.1

Type RM Length L Ch R = 1 ,291584  ,514.4,497,483.8
XS GIS Cut Line= 3
     2291409.614      528324.7282290932.67925731527651.722654008
2290613.42427293      527585.796
#Sta/Elev= 30
       0 2602.21    43.7 2574.88    97.5  2543.7   136.7 2526.76   151.4 2522.25
   210.2 2519.69   272.3 2519.33   320.7  2521.1   336.4 2520.64   359.4 2517.37
   379.4 2510.84   389.9 2509.32   528.3 2509.34   537.3 2510.87   553.4 2517.37
   560.2 2518.83     715 2516.09     805 2516.61     854 2515.34   866.2 2512.19
   878.5 2512.36   890.7 2514.18     903 2518.62   925.2 2517.61     952 2519.56
   972.4 2528.59   988.8  2537.8  1017.3 2555.57  1041.9 2572.89  1150.9 2638.16
#Mann= 7 ,-1,0
       0      .1       0     320    .025       0   379.4    .035       0
   537.3    .025       0     570      .1       0     690     .07       0
     730      .1       0
Bank Sta=379.4,537.3
XS Rating Curve= 0 ,0
Exp/Cntr=0.3,0.1

Type RM Length L Ch R = 1 ,291087  ,527.2,499.5,467
XS GIS Cut Line= 4
     2291867.629      527965.855     2291539.674      527650.484
2291313.42726528 527430.021282282290648.01978557527404.567723082
#Sta/Elev= 30
       0 2651.33   104.7 2601.62   189.6 2548.39   226.4 2528.86   254.5 2520.24
   312.6 2516.93   341.5 2518.14   367.9 2512.38     382 2511.04   404.3 2508.88
   491.2 2508.88   506.5 2511.09   523.4  2512.2   548.6 2517.81   647.9    2516
   776.1  2518.3   896.3 2515.84   984.3 2516.32  1052.3 2513.89  1208.5 2515.22
  1224.5 2511.08  1244.5 2512.75  1260.5 2517.63  1284.5 2515.93  1296.5 2518.38
  1344.6 2549.99    1354 2562.22  1380.6 2587.06  1401.3 2602.09  1436.8 2623.64
#Mann= 8 ,-1,0
       0      .1       0     382    .035       0   506.5      .1       0
  674.99     .07       0  714.99     .08       0  800.88     .07       0
  900.88     .05       0 1100.88      .1       0
Bank Sta=382,506.5
XS Rating Curve= 0 ,0
Exp/Cntr=0.3,0.1

Type RM Length L Ch R = 1 ,290587  ,539.3,501.4,461.1
XS GIS Cut Line= 3
     2292272.278      527456.364 2291547.1776246527128.796592431
2290628.74943865527210.820863533
#Sta/Elev= 30
       0 2691.94    87.1 2667.88   165.7 2623.29   226.2 2595.97   253.4 2588.34
   285.4 2583.76   307.4 2575.28   368.8 2538.88   386.4 2523.37   395.1 2511.81
   408.3 2508.43   504.4 2508.48   534.6 2511.67   561.9 2516.28   607.2 2513.53
   883.6 2517.11  1047.7 2512.63  1141.6  2515.1  1368.9 2512.19  1525.6 2514.46
  1541.6 2510.94  1561.7 2510.92  1577.8 2516.39  1593.8  2515.1  1617.9 2527.25
  1646.7 2550.43  1658.4  2567.5  1674.1 2579.91  1698.2 2592.65  1717.7 2593.62
#Mann= 10 ,-1,0
       0      .1       0     330    .025       0   395.1    .035       0
   534.6      .1       0     650     .08       0     680     .07       0
     760     .08       0  965.66      .1       0 1055.66     .05       0
 1455.66      .1       0
Bank Sta=395.1,534.6
XS Rating Curve= 0 ,0
Exp/Cntr=0.3,0.1

Type RM Length L Ch R = 1 ,290086  ,572.2,494.8,415.5
XS GIS Cut Line= 3
     2292456.301      526801.9972291551.69806647526784.603809925
 2290542.9980173527100.190904736
#Sta/Elev= 30
       0 2693.44    24.5 2681.24   212.9 2562.22   240.2 2551.53   272.2 2544.98
   292.2 2529.76   324.2 2519.06   340.2 2518.66   356.2 2512.03   372.2 2510.88
     395 2507.88   484.2 2507.84   528.2 2510.38   592.2 2514.33   744.3  2511.2
   925.2 2513.73  1222.8 2510.78  1319.2 2513.78  1646.1 2511.48  1729.9 2514.25
  1742.5 2510.34  1763.5 2510.62  1776.4  2515.4    1797 2514.27  1821.1 2524.68
  1851.5 2545.61  1864.1 2567.68  1872.4 2576.28  1922.7 2601.11  1961.7 2614.86
#Mann= 7 ,-1,0
       0      .1       0   372.2    .035       0   528.2      .1       0
     580     .05       0     680     .07       0     880     .05       0
 1594.77      .1       0
Bank Sta=372.2,528.2
XS Rating Curve= 0 ,0
Exp/Cntr=0.3,0.1

Type RM Length L Ch R = 1 ,289591  ,540.8,503.6,463.2
XS GIS Cut Line= 3
     2292124.341      526049.3842291498.98167423526642.017493635
2290515.70617015527054.633603006
#Sta/Elev= 30
       0 2549.77    87.7 2547.74     337  2536.7   342.8  2534.7   362.1 2514.57
  369.21 2508.97   377.7 2507.06     498 2507.11  541.66 2508.97   602.6 2512.65
   647.9 2510.65   918.1 2512.75  1007.8 2511.32  1085.8 2512.55  1176.9 2510.64
  1260.3 2513.22  1341.8  2512.2  1406.8 2513.84  1624.4 2511.41  1688.1 2513.91
  1701.8 2510.66  1727.9 2510.66  1740.9 2514.75  1758.4 2515.03  1779.8 2525.47
  1807.3 2549.24    1850 2589.72  1865.3 2601.02  1888.4  2612.7  1927.9 2622.29
#Mann= 10 ,-1,0
       0      .1       0     340    .025       0     360      .1       0
  369.21    .035       0  541.66    .025       0     610      .1       0
     640     .08       0     750     .05       0 1521.56     .08       0
 1631.56      .1       0
Bank Sta=369.21,541.66
XS Rating Curve= 0 ,0
Exp/Cntr=0.3,0.1

Type RM Length L Ch R = 1 ,289088  ,523.8,495.1,456.7
XS GIS Cut Line= 3
2291704.98411911525392.1791379672291239.16294639526381.833487367
 2290515.8060873 527025.23384669
#Sta/Elev= 30
       0 2603.44    48.9 2576.66    71.8 2567.39   163.7 2550.14   253.9 2537.33
   328.3 2512.41   368.2 2508.94   626.8 2511.27     651  2506.3   686.4 2507.28
   837.8 2505.97   847.2 2507.48   876.5 2509.27   889.7 2506.82   907.4 2510.62
  1041.4 2508.29    1071 2510.56  1231.6 2509.28  1571.4 2512.92    1785 2510.83
  1837.8  2512.9  1869.2 2509.76  1888.8 2514.95  1902.9 2514.54  1925.6 2525.36
  1956.8 2549.19  1991.8 2582.28  2013.4 2598.26  2030.4 2607.45  2061.9 2615.34
#Mann= 7 ,-1,0
       0      .1       0     670     .07       0   686.4    .035       0
   847.2    .025       0     890     .07       0    1000     .05       0
  1703.8      .1       0
Bank Sta=686.4,847.2
XS Rating Curve= 0 ,0
Exp/Cntr=0.3,0.1

Type RM Length L Ch R = 1 ,288593  ,514.1,498.3,480.5
XS GIS Cut Line= 3
2291003.17755782525122.968752332 2290867.6147243526367.300576493
2290469.44280196526957.372594585
#Sta/Elev= 30
       0 2614.01    78.7 2581.42   118.9 2566.74   163.2 2556.84   219.5 2541.19
   258.7 2519.11   271.8 2513.71     308 2505.76   348.3 2506.87   376.4 2503.02
   432.9 2507.59     650 2508.49   694.3 2508.08   710.4 2505.31   734.5 2505.27
  897.212505.528   903.5 2508.16   963.9 2506.09     980  2508.3  1049.7 2506.44
  1108.7 2509.34  1198.5 2509.13  1345.6 2512.22  1500.1 2510.29  1770.3 2511.58
  1805.8 2514.87  1834.7 2527.17    1875 2550.17  1910.2 2567.85  1963.5 2587.01
#Mann= 8 ,-1,0
       0      .1       0     590     .08       0   734.5    .035       0
  897.21    .025       0     980      .1       0    1080     .05       0
 1641.69     .08       0 1731.69      .1       0
Bank Sta=734.5,897.21
XS Rating Curve= 0 ,0
Exp/Cntr=0.3,0.1

Type RM Length L Ch R = 1 ,288094  ,343.2,414.8,472.9
XS GIS Cut Line= 3
2290382.32821489 525243.138045642290438.67076596 526295.00665093
 2290196.7954506526776.326603006
#Sta/Elev= 30
       0 2568.88    38.1 2557.62    75.9 2541.58    98.2    2538   102.2 2536.04
   130.2 2508.89   142.2 2502.38   170.3 2501.66   190.3 2504.51   286.5 2505.78
   430.7 2504.97   570.9 2506.49   586.9 2504.41   598.9 2502.31   751.1 2502.38
  757.73 2504.56   767.1 2505.93   843.2    2505   863.3 2507.11   967.4 2509.55
  1140.9 2508.32  1337.8 2510.92  1351.3 2508.73  1373.7 2509.18  1391.6 2513.67
  1409.5 2510.35  1427.4  2516.5  1472.1 2552.92  1524.6 2586.59  1592.1 2621.65
#Mann= 9 ,-1,0
       0      .1       0     370     .08       0     460      .1       0
     560    .025       0   586.9    .035       0  757.73    .025       0
   767.1     .05       0 1053.38     .08       0 1273.38      .1       0
#XS Ineff= 2 , 0
                         1390.87         2524.62
Permanent Ineff=
       F       F
Bank Sta=586.9,757.73
XS Rating Curve= 0 ,0
Exp/Cntr=0.3,0.1

Type RM Length L Ch R = 1 ,287679  ,649.5,624.2,582.3
XS GIS Cut Line= 3
2290225.89003722525229.511413384  2290122.987291525743.163019127
2289662.45634293526271.035801503
#Sta/Elev= 30
       0 2574.64    43.3 2564.94    85.3 2552.05   135.1 2509.58   146.5 2501.59
   150.6 2500.81   199.6 2502.54     220 2501.11   232.2 2504.47   268.9 2500.53
   289.3 2502.71   327.4 2500.62   342.3 2503.82   368.2 2504.57   547.1 2504.65
     618 2501.97   637.8 2500.03   717.6 2499.94   731.4    2502   739.9 2508.18
   745.6 2509.29   887.3 2506.65   951.2 2507.37  1025.5 2504.29  1083.9  2505.7
  1105.1 2511.84  1122.6 2510.35  1130.5 2513.64  1173.1 2546.15  1224.4 2576.54
#Mann= 8 ,-1,0
       0      .1       0     390     .08       0  603.86    .025       0
     618    .035       0   731.4     .05       0  733.86     .08       0
  853.86     .05       0  993.86      .1       0
#XS Ineff= 2 , 0
                          1105.8         2520.83
Permanent Ineff=
       F       F
Bank Sta=618,731.4
XS Rating Curve= 0 ,0
Exp/Cntr=0.3,0.1

Type RM Length L Ch R = 1 ,287055  ,464,454.1,429.4
XS GIS Cut Line= 2
2289780.91113647524981.6724545872289340.50768188526123.748119623
#Sta/Elev= 30
       0 2714.19    33.8 2701.64    46.6  2689.7    55.9 2686.31    68.1  2674.1
   133.2 2633.88   201.3 2593.87   266.3 2559.88   303.9 2542.94   342.4 2508.33
   368.4 2500.18   376.7  2497.9   470.5 2497.84   509.6 2499.48     570 2501.24
   719.7 2501.51     754 2499.22   766.9 2502.13     784 2502.12   804.6 2499.53
   832.5 2504.27   916.9 2502.35  1019.8 2511.05  1032.7 2510.38  1037.6 2512.25
  1049.8 2522.11  1062.7 2527.28  1084.1 2539.74  1174.1 2579.74    1224 2604.22
#Mann= 6 ,-1,0
       0      .1       0   368.4    .035       0   509.6      .1       0
     570     .08       0     880     .07       0     990      .1       0
#XS Ineff= 2 , 0
                         1019.04         2531.03
Permanent Ineff=
       F       F
Bank Sta=368.4,509.6
XS Rating Curve= 0 ,0
Exp/Cntr=0.3,0.1

Type RM Length L Ch R = 1 ,286601  ,130.8,178.4,252.5
XS GIS Cut Line= 4
2289352.48469827525072.3084461652289197.62504378 525258.79371785
2289132.56051077 525617.853548152288984.54428932525906.266305714
#Sta/Elev= 30
       0 2653.03    32.1 2640.03    75.6 2616.17   182.1 2567.96   199.7 2557.62
   225.2 2538.68   242.3    2528   265.2 2507.44   273.3 2504.53   281.4 2497.88
   289.5 2495.91   411.5 2496.16   419.6 2497.87   435.9 2500.98   472.5 2500.89
   525.3 2496.77   553.8 2499.78   574.1 2498.82   594.4 2501.69   651.5 2500.65
   690.3    2510     701 2509.09   714.5 2505.17   731.9  2505.9   755.7 2511.79
   768.4 2517.38   783.4 2518.53   808.9 2530.14   847.8 2550.62   931.5 2603.62
#Mann= 7 ,-1,0
       0      .1       0     210    .025       0   281.4    .035       0
   419.6     .08       0   602.4     .07       0  637.31     .08       0
  707.31      .1       0
#XS Ineff= 2 , 0
                          692.39         2526.58
Permanent Ineff=
       F       F
Bank Sta=281.4,419.6
XS Rating Curve= 0 ,0
Exp/Cntr=0.3,0.1

Type RM Length L Ch R = 1 ,286423  ,221.4,224.4,233.3
XS GIS Cut Line= 3
2289215.93920272525078.6896421612288731.35178102525638.708124788
2288699.35072487525833.000251413
#Sta/Elev= 30
       0 2613.57    24.3  2602.1    48.5 2593.02    61.5 2582.93   103.7 2562.38
     125 2556.52   140.6 2549.79     183 2525.48   211.4 2504.33   225.8 2499.86
   251.9 2496.61   262.5 2495.34   439.8 2495.19     444 2496.51   449.7 2498.25
   463.5 2497.43   486.5 2499.83   509.2 2506.81   542.8 2505.01   553.4 2508.45
     564 2508.98   590.4 2506.11   623.2 2507.16   662.3 2515.04   779.6 2527.97
   824.2 2543.04   872.8 2568.17   888.2 2584.88   921.4 2603.65   937.5  2619.6
#Mann= 4 ,-1,0
       0      .1       0   251.9    .035       0     444     .08       0
     570      .1       0
#XS Ineff= 2 , 0
                           566.2         2523.09
Permanent Ineff=
       F       F
Bank Sta=251.9,444
XS Rating Curve= 0 ,0
Exp/Cntr(USF)=0,0
Exp/Cntr=0.3,0.1

Type RM Length L Ch R = 1 ,286198  ,389.6,374.1,342.3
XS GIS Cut Line= 3
2289119.93603427524923.2559408612288509.63017769525485.560213213
2288310.76647162525556.419694688
#Sta/Elev= 30
       0  2611.5   100.3 2588.91   120.1 2582.99   168.3 2564.41   173.9 2561.83
   182.4 2554.43   191.7 2542.88   206.4 2534.15   217.2 2525.28   250.3 2509.13
   275.8 2504.17   309.7 2494.72   343.7 2497.09   360.7 2496.07   469.2  2494.5
   478.3 2496.36   494.6 2499.62   510.9 2498.21   612.6 2503.51   646.3 2507.32
   658.1 2513.47     685 2517.86   846.1  2524.8   882.4 2530.25     909 2540.27
   941.8 2557.15   984.3 2586.49    1014 2609.69  1027.9 2622.83    1041 2631.49
#Mann= 6 ,-1,0
       0      .1       0     280    .025       0   360.7    .035       0
   478.3      .1       0     540     .08       0     670      .1       0
Bank Sta=360.7,478.3
XS Rating Curve= 0 ,0
Exp/Cntr(USF)=0,0
Exp/Cntr=0.3,0.1

Type RM Length L Ch R = 1 ,285824  ,306.8,382.7,447.7
XS GIS Cut Line= 4
2288998.78917885 524703.820127262288596.49018725524868.396987461
2288438.77069622525122.1196469362288153.04698059525268.410189337
#Sta/Elev= 30
       0 2599.53    28.8 2590.43    73.6 2582.13   162.7  2560.2   223.9 2543.75
   257.6  2530.4     301 2508.71   318.3 2503.13   339.9 2501.52   355.8 2501.98
   371.1 2499.75   423.2 2500.47   426.3  2500.2   435.3 2494.95   440.3 2493.23
   458.7 2493.19   652.2 2493.26  659.62 2495.04   673.6 2498.02     708 2498.41
   727.6 2496.14   740.8 2496.34   754.3  2499.6   767.3 2506.47   785.8 2507.27
   826.2 2524.56   893.6 2543.63   918.9 2554.64   951.6 2572.62  1054.4 2636.09
#Mann= 4 ,-1,0
       0      .1       0   435.3    .035       0  659.62     .08       0
  743.41      .1       0
#XS Ineff= 2 , 0
                          772.73         2518.59
Permanent Ineff=
       F       F
Bank Sta=435.3,659.62
XS Rating Curve= 0 ,0
Exp/Cntr(USF)=0,0
Exp/Cntr=0.3,0.1

Type RM Length L Ch R = 1 ,285442  ,343.9,378,401
XS GIS Cut Line= 3
2288819.28683333524547.9034498072288530.11113108524656.344338152
2287836.08944567524837.079152061
#Sta/Elev= 30
       0 2566.96    46.9 2557.68   158.8 2529.45   180.9  2521.6   212.7 2506.91
   238.3 2498.94   251.1 2498.09     281 2500.45   343.9 2501.78     357 2501.32
   372.8 2498.42   405.4 2498.68   430.7 2502.76   451.4 2500.54   465.2 2496.88
   509.2    2494   547.2 2491.62   641.5  2491.5   649.8 2491.53   655.4 2494.04
   671.8 2504.29   682.8 2506.89   695.2 2506.76   699.4 2508.72     724 2527.23
   757.2 2559.11   786.2 2569.01   794.4 2576.15   925.2 2650.96    1026 2711.78
#Mann= 4 ,-1,0
       0      .1       0  408.84     .08       0   509.2    .035       0
   655.4      .1       0
Bank Sta=509.2,655.4
XS Rating Curve= 0 ,0
Exp/Cntr(USF)=0,0
Exp/Cntr=0.3,0.1

Type RM Length L Ch R = 1 ,285064  ,288.4,280.1,267
BEGIN DESCRIPTION:
c/e of 0.5/0.7 used to correct drawdown in the 100 year profile
END DESCRIPTION:
XS GIS Cut Line= 2
     2288699.974      524389.874     2287790.292      524324.396
#Sta/Elev= 30
       0 2549.98      60 2536.87   156.2 2503.18   204.3 2497.14   232.4 2495.78
   296.6 2500.14   356.7 2499.75   399.7 2492.45   408.9 2490.41   509.1 2490.44
  514.572492.542   525.2 2501.08   533.2 2504.73   573.3 2505.18   581.3 2512.68
   589.3 2523.28   593.3 2525.65   610.3 2527.95   642.9    2540   677.6 2548.15
   725.7  2573.7   744.9 2593.85   769.8 2614.03   781.8 2621.39   817.9 2651.04
   829.9 2665.78     842 2676.05     862 2698.75   882.1 2716.18     912  2750.6
#Mann= 3 ,0,0
       0      .1       0   399.7    .035       0  514.57      .1       0
Bank Sta=399.7,514.57
XS Rating Curve= 0 ,0
Exp/Cntr=0.7,0.5

Type RM Length L Ch R = 1 ,284783  ,345.4,369.2,394.1
BEGIN DESCRIPTION:
IFA added to correct drawdown
END DESCRIPTION:
XS GIS Cut Line= 3
2288678.25536804524055.8384617822288101.46973804 524089.11455582
2287805.15404351524073.268796754
#Sta/Elev= 30
       0 2568.65    38.1 2557.45   102.3 2526.61   130.3  2511.2   158.3 2499.76
   204.9  2497.4   230.5 2494.34   243.1 2495.95   262.5 2495.15   274.5 2496.79
   302.5 2495.41   346.7 2496.51  356.85 2491.08   362.7 2489.06     440 2489.09
   456.22489.125   514.9 2489.16   522.2 2490.83     543  2500.5     551 2502.65
     559  2502.7   591.1 2524.11   611.1 2534.05   659.6 2566.02   707.2 2594.55
   783.3 2636.82   823.4  2663.2   847.4 2685.56   859.4 2695.07   874.5 2709.83
#Mann= 5 ,-1,0
       0      .1       0  356.85    .035       0     440     .08       0
   456.2    .035       0   522.2      .1       0
#XS Ineff= 2 , 0
          319.44 2516.33
Permanent Ineff=
       F       F
Bank Sta=356.85,522.2
XS Rating Curve= 0 ,0
Exp/Cntr(USF)=0,0
Exp/Cntr=0.3,0.1

Type RM Length L Ch R = 1 ,284414  ,309,315.9,322.7
XS GIS Cut Line= 2
 2288747.3523091523858.0779290082287910.75326974523620.355797608
#Sta/Elev= 30
       0 2589.27    45.4 2573.51    97.2 2552.32   190.4 2503.57   202.9 2499.39
   219.5 2496.53   248.6 2495.41   273.6 2492.44   302.7 2494.65   356.8 2495.69
   406.7 2492.64   448.2 2493.47   464.9 2491.86   479.3 2487.93   498.7 2485.81
   560.3 2485.65   568.8 2486.03     573  2488.1   593.8 2498.05   606.3  2501.2
   614.6 2505.85   627.1 2529.29   635.4 2538.06   663.9 2559.11   701.9  2594.5
   805.9 2678.03   819.3 2693.22   847.4 2712.04   855.8 2720.25   869.7 2730.44
#Mann= 3 ,0,0
       0      .1       0   479.3    .035       0     573      .1       0
Bank Sta=479.3,573
XS Rating Curve= 0 ,0
Exp/Cntr(USF)=0,0
Exp/Cntr=0.3,0.1

Type RM Length L Ch R = 1 ,284098  ,506.1,508.9,512
XS GIS Cut Line= 2
2288850.99553301523615.476747895     2287931.016      523253.067
#Sta/Elev= 30
       0 2594.83    41.7 2579.27   139.7 2537.37   182.8 2512.64     218 2496.69
   256.7 2494.28   334.1 2495.09   394.3 2490.64   441.9 2492.89   472.7 2490.73
   483.3 2487.34   497.4 2484.62     592 2484.66   599.2 2487.03   611.5 2494.93
   626.4 2500.16   630.7 2506.87   639.3 2525.71   647.9 2535.37   679.4 2559.31
   707.1 2584.09   742.5 2611.74   813.9 2664.03   841.4 2688.05   929.2  2770.7
   940.3 2779.43   944.6 2785.05   953.1 2804.01     957 2810.08   988.8 2839.64
#Mann= 4 ,-1,0
       0      .1       0     450     .07       0   483.3    .035       0
   599.2      .1       0
Bank Sta=483.3,599.2
XS Rating Curve= 0 ,0
Exp/Cntr=0.3,0.1

Type RM Length L Ch R = 1 ,283589  ,443.5,452.8,460.4
XS GIS Cut Line= 2
2289114.71983872523199.850723082      2288123.55      522762.303
#Sta/Elev= 30
       0 2589.23    31.3 2579.31      95 2554.42   179.8 2510.83   210.2 2497.68
   219.3 2495.08   265.1 2493.15     405 2493.32   495.4 2490.71   516.4 2491.28
   523.1  2490.4   534.6 2485.71     545 2483.56   676.1 2483.56   684.9  2485.4
   702.4 2495.56   719.9 2497.99     732 2513.36     738 2526.87   747.1 2541.39
   754.8 2549.43   772.3  2564.1   794.2 2595.23   798.2 2599.53   824.8 2616.99
   856.3 2634.28   894.8 2650.72   942.9 2661.42   986.6 2674.01  1083.5 2691.56
#Mann= 5 ,-1,0
       0      .1       0     530    .025       0   534.6    .035       0
   684.9    .025       0     750      .1       0
Bank Sta=534.6,684.9
XS Rating Curve= 0 ,0
Exp/Cntr=0.3,0.1

Type RM Length L Ch R = 1 ,283137  ,533.3,544.2,552.3
XS GIS Cut Line= 3
2289507.37724788522878.6911871612289202.92936213522796.664286712
2288328.73440984522312.960590159
#Sta/Elev= 30
       0 2590.75    82.2 2572.31     140  2555.4   181.5 2539.33     227 2516.92
   239.4 2513.23   432.7 2492.78   697.9 2491.55     739 2487.78   761.4 2489.64
     771 2484.91   780.2 2483.09   908.2  2483.1   920.3 2485.22   940.2 2495.91
   953.9 2494.41   958.5 2497.02   966.9 2508.99  1002.7 2539.96  1016.5 2559.19
    1027  2571.5  1045.3 2585.65  1072.7 2602.89  1117.5 2637.13  1132.2 2662.13
  1176.3 2690.54  1191.6 2696.75  1211.6 2698.57  1252.8  2697.1  1314.4 2689.65
#Mann= 6 ,-1,0
       0      .1       0   525.3     .12       0   635.3      .1       0
   745.3     .12       0     771    .035       0   920.3      .1       0
Bank Sta=771,920.3
XS Rating Curve= 0 ,0
Exp/Cntr=0.3,0.1

Type RM Length L Ch R = 1 ,282592  ,411,415.1,418.5
XS GIS Cut Line= 3
2289649.42090474522496.5853965412288785.54966807521923.633951844
 2288475.7947315521881.523913158
#Sta/Elev= 30
       0 2570.12    40.9 2559.47    78.4 2547.07   174.3 2496.04   342.3 2491.44
     520 2489.38   539.1 2489.99   582.3 2486.69   601.5 2490.27   683.1 2490.19
   690.7 2485.61   697.5 2482.56     872  2482.6   879.9 2485.22   884.7 2488.69
   889.5 2489.12     918 2482.89   932.5 2483.34   951.9  2490.1   995.1 2488.92
  1028.7 2493.03  1046.1 2492.94  1062.2 2505.18  1122.8 2535.83  1163.1 2559.26
  1223.7 2599.04  1246.1 2623.07  1296.3  2659.5  1331.4 2680.84  1349.2 2687.01
#Mann= 7 ,-1,0
       0      .1       0     440     .08       0     520      .1       0
     620     .08       0     640    .025       0   690.7    .035       0
   879.9      .1       0
#XS Ineff= 2 , 0
           440.9 2511.56 1027.72         2512.81
Permanent Ineff=
       F       F
Bank Sta=690.7,879.9
XS Rating Curve= 0 ,0
Exp/Cntr=0.3,0.1

Type RM Length L Ch R = 1 ,282177  ,599,566.1,552.7
XS GIS Cut Line= 4
2289865.10348462521917.4424524782289471.94765192521894.584555228
2289133.65077262521652.2908443772288402.19806062521702.578218328
#Sta/Elev= 30
       0  2554.3    81.1 2528.74     145 2512.31   166.6 2508.88   233.3 2505.92
   289.4 2500.58   460.6 2494.24   477.2 2491.96   497.9 2483.46   595.3 2488.37
  613.24 2483.88   622.9 2482.12   762.5 2482.16   772.4 2483.73   793.2 2488.24
   983.8 2489.53    1068 2489.09  1108.1 2482.61  1144.2 2484.97  1179.8 2483.21
  1192.3  2485.3  1204.3 2491.34  1228.4 2491.35  1252.5 2507.91  1380.8  2574.9
  1440.9 2614.92    1473 2634.23    1485 2638.09  1498.7 2638.45  1543.1 2630.79
#Mann= 5 ,-1,0
       0      .1       0  583.82     .08       0  613.24    .035       0
   772.4     .12       0  793.82      .1       0
#XS Ineff= 2 , 0
                         1206.99          2499.7
Permanent Ineff=
       F       F
Bank Sta=613.24,772.4
XS Rating Curve= 0 ,0
Exp/Cntr(USF)=0,0
Exp/Cntr=0.3,0.1

Type RM Length L Ch R = 1 ,281611  ,629.9,496.8,417
XS GIS Cut Line= 4
     2289964.356      521479.0342289386.67561587521177.983884361
2289216.02674737521089.6384106282288493.52811568521447.489791956
#Sta/Elev= 30
       0 2526.23    36.3 2526.15    73.3 2523.25    90.5 2519.71   133.8 2505.98
   248.3 2497.74   253.6 2496.47   266.3 2486.58   275.3 2482.71   288.9 2479.94
   478.3 2479.97   502.6 2482.66   517.5 2483.42   529.3 2486.81   703.8 2485.21
   834.4 2487.02  1008.6 2485.73  1121.9 2488.19    1270 2487.38  1383.4 2483.69
  1459.4 2485.27  1490.7 2479.44  1502.9 2482.92  1514.8 2489.66  1530.8  2489.4
  1535.3 2491.32  1544.6 2499.27  1562.1 2505.64  1583.5  2516.3  1649.8 2556.12
#Mann= 3 ,-1,0
       0      .1       0   275.3    .035       0   502.6      .1       0
#XS Ineff= 2 , 0
                         1513.01         2499.07
Permanent Ineff=
       F       F
Bank Sta=275.3,502.6
XS Rating Curve= 0 ,0
Exp/Cntr=0.3,0.1

Type RM Length L Ch R = 1 ,281114  ,227.9,222.2,217.2
XS GIS Cut Line= 2
2290117.87182632520535.1894793992288504.63348384521384.375536992
#Sta/Elev= 30
       0    2523      56 2515.52    96.8  2503.8     176 2491.04   390.7 2489.03
   425.1 2486.21   440.4 2488.96   485.6 2489.22   503.2 2480.43   523.9 2481.41
   532.8 2479.25   634.8 2479.17   648.3 2481.25   680.9 2483.56     717 2481.56
     760 2483.03   787.5 2479.45   811.2 2483.78   874.3 2482.53   914.9 2486.88
   964.7 2484.46  1308.3 2488.13  1529.8 2484.18  1665.4 2484.78    1696 2479.29
  1714.4 2483.17  1726.3 2489.74  1742.2 2489.25  1764.7 2502.02  1823.1 2528.31
#Mann= 3 ,0,0
       0      .1       0   523.9    .035       0   648.3      .1       0
#XS Ineff= 2 , 0
          460.85 2498.42
Permanent Ineff=
       F       F
Bank Sta=523.9,648.3
XS Rating Curve= 0 ,0
Exp/Cntr=0.3,0.1

Type RM Length L Ch R = 1 ,280892  ,785.7,754.9,765.2
XS GIS Cut Line= 3
 2289999.9650784520296.8175374492289252.51183832520765.404431075
2288434.19911677521249.991852776
#Sta/Elev= 30
       0 2527.91   131.9 2513.03   182.9 2494.12     198 2491.62   245.2 2488.24
   419.9 2488.13   471.9 2480.25   525.3 2483.99   542.8 2482.86   547.1 2480.46
   658.8  2478.8   673.3 2480.44   783.9 2481.42   866.7 2477.81   889.6 2481.83
   917.3 2483.21  1045.3 2478.27  1060.4 2484.13  1110.4  2485.6  1235.6  2483.1
  1273.5 2485.49    1548 2482.55  1598.5 2483.92  1626.4 2479.71  1686.8 2479.46
  1714.7 2488.45  1742.6 2489.15  1756.5 2497.81  1804.9 2519.77  1833.2 2530.01
#Mann= 3 ,0,0
       0      .1       0   547.1    .035       0   673.3      .1       0
#XS Ineff= 2 , 0
          413.52 2499.64
Permanent Ineff=
       F       F
Bank Sta=547.1,673.3
XS Rating Curve= 0 ,0
Exp/Cntr(USF)=0,0
Exp/Cntr=0.3,0.1

Type RM Length L Ch R = 1 ,280137  ,582.1,611,451.7
XS GIS Cut Line= 2
2289628.97879965 519762.04557749 2288173.4610983521060.926440118
#Sta/Elev= 30
       0 2523.91    86.9 2506.98   102.9 2498.68   124.4 2492.95   161.9 2492.09
   199.4 2503.23   277.6 2499.79   305.1 2481.62   345.6 2475.23   464.6 2479.78
   575.4 2477.46   735.6 2481.33   762.4 2476.84   791.7 2481.12   881.8 2483.58
   929.9  2479.5  1068.1 2480.16  1105.5 2477.32  1201.1 2475.16  1232.3 2477.58
  1242.3  2482.8  1512.8 2479.63  1604.1 2482.97  1644.8 2475.89  1695.2 2476.15
  1730.9 2487.29  1750.7 2487.53  1793.2 2520.45    1837 2547.69  1950.8 2592.35
#Mann= 4 ,-1,0
       0      .1       0    1080    .025       0  1105.5    .035       0
  1232.3      .1       0
Bank Sta=1105.5,1232.3
XS Rating Curve= 0 ,0
Exp/Cntr(USF)=0,0
Exp/Cntr=0.3,0.1

Type RM Length L Ch R = 1 ,279526  ,746.9,645.8,349.2
XS GIS Cut Line= 3
2289339.80309739519648.7850941072288566.25809386520022.303709519
 2288161.4121107 521036.82846493
#Sta/Elev= 30
       0 2521.57    30.7 2517.87    70.7 2505.26   102.1 2500.12   159.5 2498.32
   186.1 2481.15   226.1 2475.43   359.7 2481.91   568.2 2478.15   641.1 2480.86
     657 2476.39   750.3 2475.62   812.5 2479.19   918.2 2474.87   933.6 2473.74
  1010.9 2475.92  1037.3 2479.61  1149.1 2478.34  1241.1 2474.18    1254 2481.31
  1322.9 2482.32  1538.3  2481.2  1570.8 2475.09  1628.7 2480.37  1723.4 2479.77
    1745 2486.96  1766.5 2487.59  1792.5 2507.85  1852.6 2543.69  1951.3 2583.41
#Mann= 6 ,-1,0
       0      .1       0     657    .035       0   750.3      .1       0
   918.2    .035       0  1010.9     .08       0  1149.1      .1       0
Bank Sta=657,1010.9
XS Rating Curve= 0 ,0
Exp/Cntr(USF)=0,0
Exp/Cntr=0.3,0.1

Type RM Length L Ch R = 1 ,278881  ,465.6,512.7,509.7
XS GIS Cut Line= 3
2288028.87324717519725.8986147082288277.08239161520405.461515007
2288139.72393303521019.959882298
#Sta/Elev= 30
       0 2541.24    79.6 2514.36   122.7 2490.06     144 2481.75   216.4 2477.73
   226.6 2475.21   250.5 2472.44   369.7 2472.68   385.7 2474.84   403.8 2477.71
   450.6 2475.28   467.7 2477.35     489 2473.43   518.8 2473.35   557.1 2477.72
   599.7 2476.46   622.7  2479.4   663.6 2478.07   723.2 2480.57   822.2 2478.22
   901.5 2480.72     924 2475.31   985.3 2475.49  1059.3 2482.07  1104.4 2481.87
  1124.9 2479.26  1149.4 2486.84  1169.5 2487.35  1260.3 2539.88  1353.1 2578.15
#Mann= 6 ,-1,0
       0      .1       0   226.6    .035       0   385.7    .025       0
     390      .1       0     500     .08       0     710      .1       0
Bank Sta=226.6,385.7
XS Rating Curve= 0 ,0
Exp/Cntr(USF)=0,0
Exp/Cntr=0.3,0.1

Type RM Length L Ch R = 1 ,278368  ,278.4,294,295.9
XS GIS Cut Line= 4
2287579.31375962519839.6595924482287666.17376917520077.381723848
2287741.60483009520356.2480702992287748.46219927520980.268665226
#Sta/Elev= 30
       0 2563.67    48.6  2543.1    86.1 2532.59   112.3  2521.3   142.2 2500.51
   154.9 2488.43   176.2 2471.93   218.8  2471.7   235.8  2476.1   248.6 2476.52
   269.5 2475.69  280.48 2472.98   290.4 2470.19   306.7 2470.06   402.1    2470
   414.4 2472.81   430.7 2474.31   437.2 2472.32     447 2470.15     509 2469.88
   526.4 2469.94  536.33 2473.11   550.9  2477.9   914.9 2479.36   942.9 2485.56
   954.9 2485.62   970.9  2494.5   981.2 2497.45  1030.9 2526.13    1166 2594.16
#Mann= 5 ,-1,0
       0      .1       0  280.48    .035       0   414.4      .1       0
   437.2    .035       0  536.33      .1       0
Bank Sta=280.48,536.33
XS Rating Curve= 0 ,0
Exp/Cntr(USF)=0,0
Exp/Cntr=0.3,0.1

Type RM Length L Ch R = 1 ,278074  ,486.2,547.4,554.1
XS GIS Cut Line= 4
2287346.16320767519908.2332841982287419.30847887520205.385948449
2287476.45322199  520575.68388392287483.31059117520971.125506326
#Sta/Elev= 30
       0 2598.37    28.9 2577.99    42.1  2564.3    66.9 2547.88   112.2 2526.17
   157.5 2510.05   169.9 2502.39   206.9 2471.81   215.2 2468.81   286.7 2470.29
     322 2472.94   338.2 2472.41   345.2 2470.31     496 2468.88   508.2 2472.05
   516.3 2475.98   564.8  2474.6   645.8 2475.87   694.2 2478.91   786.2 2478.83
   810.2 2475.62   826.2 2478.99   838.2 2483.96   854.2 2482.71   874.2 2493.89
   882.5 2495.79   914.2 2515.47   954.2 2536.74  1016.2 2565.32  1076.2 2595.55
#Mann= 5 ,-1,0
       0      .1       0   206.9    .035       0   286.7      .1       0
   345.2    .035       0   508.2      .1       0
Bank Sta=206.9,508.2
XS Rating Curve= 0 ,0
Exp/Cntr(USF)=0,0
Exp/Cntr=0.3,0.1

Type RM Length L Ch R = 1 ,277527  ,469.7,509.8,520
XS GIS Cut Line= 3
2287017.00948727519935.6627608982286925.57789827520120.811728623
2286934.72105717  520886.5512865
#Sta/Elev= 30
       0 2663.31      38  2643.7    55.2 2636.69   117.7 2600.83     140 2585.53
   155.5 2577.16   191.6 2553.96   212.3 2537.75   222.9 2532.62   234.9 2524.56
   246.9 2514.82   282.9 2491.08   305.5 2472.03   310.9 2468.12   314.9 2467.69
   394.6 2467.66   495.2 2467.63   558.9 2467.61   566.9 2467.83   573.1 2471.33
   582.9 2474.89   614.9 2473.57   718.9 2475.62     747 2477.22   774.9 2481.91
   802.9 2479.99   862.9 2516.35   878.9 2521.27   934.9 2534.27   972.3 2545.91
#Mann= 5 ,-1,0
       0      .1       0   305.5    .035       0   394.6      .1       0
   495.2    .035       0   573.1      .1       0
#XS Ineff= 2 , 0
                           764.2         2515.24
Permanent Ineff=
       F       F
Bank Sta=305.5,573.1
XS Rating Curve= 0 ,0
Exp/Cntr(USF)=0,0
Exp/Cntr=0.3,0.1

Type RM Length L Ch R = 1 ,277017  ,424.3,439.7,450
XS GIS Cut Line= 2
2286511.84995804519889.9469663982286358.70204647520824.834963925
#Sta/Elev= 30
       0 2601.38    39.8 2580.33    84.3 2554.82   144.9 2528.16     210 2491.32
   234.3 2479.16   246.3 2475.23   254.6 2474.23   327.5 2474.01   331.6 2473.54
   339.7 2468.72   343.8 2466.62   493.6 2466.22   505.9 2468.47   554.5 2471.55
   631.5 2470.02     664 2471.09   692.3 2469.51   704.5 2471.43   712.6 2476.94
   720.7 2479.63   736.9 2480.01   753.1 2489.76   765.4 2494.81   785.6 2505.96
   797.7 2514.58   809.9 2519.15     822 2528.19   907.2 2575.64   947.3 2601.48
#Mann= 4 ,-1,0
       0      .1       0   339.7    .035       0   505.9    .025       0
     510      .1       0
Bank Sta=339.7,505.9
XS Rating Curve= 0 ,0
Exp/Cntr(USF)=0,0
Exp/Cntr=0.3,0.1

Type RM Length L Ch R = 1 ,276577  ,454.7,490.1,517.3
XS GIS Cut Line= 2
2286199.90215286519857.430429775     2285846.644      520762.005
#Sta/Elev= 30
       0 2547.49    55.6 2524.12    81.3  2518.4   102.8 2518.29     120 2514.74
   158.6 2490.05   175.8  2472.9   188.7 2466.55   201.6 2469.36   227.3 2469.77
   235.9 2466.98   253.1 2470.38   313.2 2472.17   334.7 2471.04   343.3 2467.32
   360.4 2465.43   373.3 2465.31   381.9 2469.61   399.1 2470.05   447.4 2466.03
   566.6  2464.5  572.992466.122   592.3 2477.79   611.1 2480.47   652.4 2519.12
   721.2 2561.39     802 2616.39   918.7 2699.64   927.3 2709.06   971.1 2741.33
#Mann= 3 ,-1,0
       0      .1       0   447.4    .035       0  572.99      .1       0
Bank Sta=447.4,572.99
XS Rating Curve= 0 ,0
Exp/Cntr=0.3,0.1
