HEC-RAS study GRNBRRRV.prj: GRNBRRRV

--- GRNBRRRV.g01 (geometry) --- (continued)

Type RM Length L Ch R = 1 ,276087  ,491.2,500,507.2
XS GIS Cut Line= 2
      2285932.03      519709.332      2285316.06      520379.168
#Sta/Elev= 30
       0 2564.98    21.5 2559.02    86.7 2530.67   118.7 2528.03   135.7 2523.62
     198 2496.94   211.7  2489.1   222.6 2479.75   243.2 2470.37   276.9 2469.69
   320.4 2465.02   336.6 2471.08   356.5 2471.23   366.2 2469.77   374.7 2464.87
   384.8 2462.37   505.2 2462.44     515 2465.19   532.3 2474.51   548.6 2478.15
   613.9 2523.05   628.3 2540.59   764.1 2645.55   791.6 2670.12   817.9 2688.18
     833    2696   842.1 2706.59   850.7 2721.05   860.4 2729.39     910 2763.46
#Mann= 3 ,-1,0
       0      .1       0   374.7    .035       0     515      .1       0
Bank Sta=374.7,515
XS Rating Curve= 0 ,0
Exp/Cntr=0.3,0.1

Type RM Length L Ch R = 1 ,275587  ,500.6,500,499.8
XS GIS Cut Line= 2
     2285614.254      519380.995     2284938.148      519990.077
#Sta/Elev= 30
       0 2523.86      62 2513.09   131.9 2504.19     231  2498.2   245.1  2493.3
   263.2 2481.08   273.5 2477.19   298.9 2476.66   318.8 2474.29   338.6 2469.11
   372.6 2468.29   389.6 2462.93   403.8 2460.12   492.7 2460.14   502.9 2463.27
   514.2 2471.28   519.6  2473.5   545.4 2476.13   550.1 2483.93   562.7 2513.36
   579.4 2525.67   589.6 2542.82     595 2547.77   621.9 2565.96   632.7 2570.25
   686.5 2575.11   741.3 2573.18     789 2568.01   831.9 2560.64     910 2551.08
#Mann= 3 ,0,0
       0      .1       0   389.6    .035       0   502.9      .1       0
Bank Sta=389.6,502.9
XS Rating Curve= 0 ,0
Exp/Cntr=0.3,0.1

Type RM Length L Ch R = 1 ,275087  ,505.5,500,495.7
XS GIS Cut Line= 2
     2285277.154      519008.893     2284603.858      519621.079
#Sta/Elev= 30
       0 2594.32    17.5 2587.53      49 2571.34    74.5 2559.85   120.3 2543.07
   178.8 2519.49   220.4 2512.18   258.6 2494.62   284.1 2492.19   295.4 2488.95
   303.7 2485.06   327.4 2469.94     335 2467.27   363.1 2466.66   377.5 2462.33
   394.5 2458.87   482.3 2458.81   505.8 2458.86   513.4 2461.83   529.6 2466.54
   541.7 2472.17   561.6 2474.04   578.5 2484.79   592.7 2489.38   606.9 2497.44
   672.3 2540.94   752.8 2589.97   763.6 2594.27   864.5 2657.83     910  2684.8
#Mann= 7 ,-1,0
       0     .06       0      10      .1       0     130     .06       0
     150      .1       0     300     .12       0   377.5    .035       0
   513.4      .1       0
Bank Sta=377.5,513.4
XS Rating Curve= 0 ,0
Exp/Cntr=0.3,0.1

Type RM Length L Ch R = 1 ,274587  ,501.8,504.7,510.8
BEGIN DESCRIPTION:
c/e of 0.5/0.7 added to correct drawdown between the 100-500 yr events
END DESCRIPTION:
XS GIS Cut Line= 2
     2284906.619      518635.753     2284269.376      519285.385
#Sta/Elev= 30
       0 2629.18    33.9 2609.87    46.8 2601.62   130.9 2555.94   144.2 2547.53
   161.1 2534.34   172.5 2530.32   226.3 2521.67   254.5 2512.69   270.9 2505.39
   310.2 2497.24   351.9 2483.64   374.8 2469.68     383 2462.79   388.6    2459
   394.2 2457.97   511.9 2458.06     529 2463.22   537.3  2468.5   545.5 2471.16
   563.3 2469.93   585.4 2475.82   646.4 2482.69   668.8 2487.51     680 2491.52
   740.4 2518.25   763.6 2530.91   775.2 2535.06     857  2578.7     910 2609.54
#Mann= 6 ,-1,0
       0      .1       0    33.9     .06       0   172.5      .1       0
   310.2     .12       0     383    .035       0     529      .1       0
#XS Ineff= 2 , 0
       0                   548.6       0    2480
Permanent Ineff=
       F       F
Bank Sta=383,529
XS Rating Curve= 0 ,0
Exp/Cntr=0.7,0.5

Type RM Length L Ch R = 1 ,274082  ,500.9,492.2,482.4
XS GIS Cut Line= 3
     2284578.635      518292.6012284115.36207666 518706.55426426
2283667.80704564518768.567541429
#Sta/Elev= 30
       0 2635.26    36.1 2615.26    53.1 2603.85    62.3 2600.21    84.3 2587.45
   115.9 2571.68   149.5 2556.07     181 2538.74   268.4 2480.13   282.2 2473.58
     301 2468.26     313 2460.47   319.4  2457.4   325.2 2456.75   502.2 2456.86
   526.2 2459.95   548.9 2468.87   555.8  2468.5   566.5 2464.61   580.1  2472.1
   598.7 2476.75   701.6 2487.11   815.3 2488.86   875.1 2495.29   899.1 2502.87
   931.4 2518.97   979.9 2545.86   991.7  2553.9  1024.3 2570.35  1073.1  2598.2
#Mann= 5 ,-1,0
       0      .1       0      50     .06       0     250      .1       0
     313    .035       0   526.2      .1       0
#XS Ineff= 2 , 0
                          547.61         2490.95
Permanent Ineff=
       F       F
Bank Sta=313,526.2
XS Rating Curve= 0 ,0
Exp/Cntr=0.3,0.1

Type RM Length L Ch R = 1 ,273590  ,499.1,503.4,502.7
XS GIS Cut Line= 2
2284199.04141648517940.7503748962283613.68345845518542.712666844
#Sta/Elev= 30
       0 2593.58    27.1  2580.5    33.4 2576.39    44.3 2573.42    50.8 2569.31
    87.2 2552.93     101 2545.39     124 2534.68   163.6 2513.17     206 2497.33
   245.6 2476.27   257.2 2464.29  263.94 2458.96   273.9 2454.69   279.5 2454.62
   458.1 2454.75   463.4 2455.03   471.9    2459   480.3 2461.93   486.1  2462.1
   505.8 2466.44     520 2467.59   539.8 2467.55   554.9    2476   612.3 2488.47
   642.2 2496.66   686.9 2512.59   742.7 2535.59   790.2 2558.45   839.6 2583.79
#Mann= 5 ,-1,0
       0     .06       0     120      .1       0     260     .12       0
  263.94    .035       0   471.9      .1       0
Bank Sta=263.94,471.9
XS Rating Curve= 0 ,0
Exp/Cntr=0.3,0.1

Type RM Length L Ch R = 1 ,273087  ,443,495.2,543.9
XS GIS Cut Line= 3
 2284148.4707891517646.0718387212283712.92589102517732.996066669
     2283318.594      518150.812
#Sta/Elev= 30
       0 2627.17    65.6 2591.42    77.8 2582.61      86  2579.2    98.2  2571.1
   126.7 2556.98     139 2555.02   175.7 2541.43   240.9 2511.54   363.3 2470.94
   387.1 2466.65   460.9 2463.68   471.9 2460.86   480.2 2455.89   487.2 2452.84
   509.3 2452.78   637.5 2452.79   648.5 2456.03     655 2459.37   676.8 2458.04
   707.5  2464.1   736.2 2465.64   748.3 2470.16   767.4 2484.23     859 2543.76
     889  2565.9   966.9 2614.42  1010.7 2643.61  1016.4 2649.59  1018.6 2653.84
#Mann= 5 ,-1,0
       0      .1       0     150     .06       0     250      .1       0
   480.2    .035       0   648.5      .1       0
Bank Sta=480.2,648.5
XS Rating Curve= 0 ,0
Exp/Cntr=0.3,0.1

Type RM Length L Ch R = 1 ,272591  ,502.7,505.1,506
XS GIS Cut Line= 2
     2283830.561      517270.784     2282955.343      517520.133
#Sta/Elev= 30
       0 2527.01      94 2488.18   143.9 2470.26   177.2 2465.51   260.3 2461.98
     356 2460.25     381 2457.87   389.3 2454.29   397.6 2451.31   475.9 2451.28
   492.7 2451.67   500.2 2454.29   514.1 2461.49   526.5 2462.97   530.7 2467.98
   543.2  2489.9   547.3 2495.58   568.1 2515.93   576.4 2522.65   588.9 2539.86
   605.6 2555.92     618 2570.08   638.8 2586.96   709.5 2638.93   761.3 2680.27
   835.8 2744.64     851  2764.1   871.4 2784.08   880.1 2797.29     910 2815.38
#Mann= 4 ,-1,0
       0     .06       0      30      .1       0   389.3    .035       0
   500.2      .1       0
Bank Sta=389.3,500.2
XS Rating Curve= 0 ,0
Exp/Cntr=0.3,0.1

Type RM Length L Ch R = 1 ,272086  ,512,499.4,473.7
XS GIS Cut Line= 2
2283730.31284299516794.6556629532282946.10493091516989.826344725
#Sta/Elev= 30
       0 2514.86    26.9 2506.53    47.5 2497.98    79.8 2488.42   175.3 2467.12
   204.2 2462.77   248.1 2459.18   274.3 2452.63   290.7 2454.07     299 2457.81
   315.5 2458.73   336.1 2456.07   348.5 2451.29   356.7 2448.88     468 2448.94
475.93052451.199   496.8 2461.46   509.2 2462.06   533.9 2487.23   542.2 2497.03
   575.2 2523.84   579.3 2528.94   591.3 2556.98   601.3 2575.19     604 2579.18
   616.4 2590.34   687.1 2640.72   756.5 2693.08   793.6  2716.7   808.1 2724.32
#Mann= 4 ,-1,0
       0     .06       0      30      .1       0   348.5    .035       0
475.9305      .1       0
Bank Sta=348.5,475.9305
XS Rating Curve= 0 ,0
Exp/Cntr=0.3,0.1

Type RM Length L Ch R = 1 ,271587  ,495.5,500,509.1
XS GIS Cut Line= 2
     2283645.429      516209.784     2282827.474      516608.596
#Sta/Elev= 30
       0 2582.87    63.3 2556.59    99.3 2547.08   130.4 2544.19   152.7 2543.94
   162.9 2541.08     174 2535.81   191.9 2532.82   210.6 2524.58   241.7 2505.41
   260.7 2495.69     304 2485.11   366.3 2477.25   386.4 2469.08   400.2 2456.06
   406.4 2451.72   415.3 2447.38   482.4 2447.22   539.9 2450.21   547.9 2451.89
   562.9 2458.76   571.9 2460.47   584.4 2459.92   597.7 2468.15   631.7 2485.49
   652.6 2499.32   717.9 2536.51   810.9 2595.93   882.5  2638.2     910 2653.05
#Mann= 5 ,-1,0
       0      .1       0     100     .06       0     260      .1       0
   406.4    .035       0   547.9      .1       0
Bank Sta=406.4,547.9
XS Rating Curve= 0 ,0
Exp/Cntr=0.3,0.1

Type RM Length L Ch R = 1 ,271087  ,506.3,500,494.2
XS GIS Cut Line= 2
     2283469.482      515779.978     2282623.165      516114.414
#Sta/Elev= 30
       0 2548.56    87.4 2544.59   104.6 2542.52   130.4 2536.72   173.4 2521.35
   205.4 2504.68   246.6  2497.2   272.4  2490.2   285.3 2485.53   293.9 2484.15
   311.1 2478.11   347.2 2461.18   362.7 2456.81   375.6  2449.1   379.9 2446.67
   384.2 2446.28   513.2 2446.28   522.9 2448.51   532.2 2453.14     539 2457.87
   543.3 2459.21   556.2 2460.45   573.4 2474.42   586.3 2483.15   677.1 2535.07
   706.8 2553.95   723.3 2565.32   745.5 2584.37     818  2635.1     910 2702.87
#Mann= 4 ,-1,0
       0     .06       0     170      .1       0   375.6    .035       0
   522.9      .1       0
Bank Sta=375.6,522.9
XS Rating Curve= 0 ,0
Exp/Cntr=0.3,0.1

Type RM Length L Ch R = 1 ,270587  ,492,502.6,513.1
XS GIS Cut Line= 2
     2283261.828      515292.041     2282439.863      515682.519
#Sta/Elev= 30
       0 2581.19    28.4 2578.43    80.2 2576.94   103.7  2570.6   179.2 2535.58
   218.3 2524.39   266.3 2507.07   293.3 2493.44   332.3 2478.38   347.6  2475.5
   359.4 2468.78   384.9 2447.97   392.4 2444.38   413.4 2444.03   488.5 2444.12
     520 2447.84   537.7 2457.05   548.5 2458.55   564.2 2457.72   626.6 2491.17
   679.4 2524.67   683.6 2529.43   688.2 2537.35   697.1 2544.04   705.9 2567.08
   710.6 2572.93   745.8 2585.15   772.4 2597.24   891.9 2665.33     910 2678.27
#Mann= 4 ,-1,0
       0     .06       0     160      .1       0   384.9    .035       0
     520      .1       0
Bank Sta=384.9,520
XS Rating Curve= 0 ,0
Exp/Cntr=0.3,0.1

Type RM Length L Ch R = 1 ,270084  ,491.5,498.3,505.5
XS GIS Cut Line= 2
     2283083.925      514888.945     2282216.679      515164.741
#Sta/Elev= 30
       0 2574.02    58.5 2548.99   105.1 2524.76   129.9  2515.8   142.4 2513.89
     176 2496.72   213.4 2482.51   251.5 2465.05   299.3  2453.5   385.9 2449.72
   399.3 2446.15   427.9 2442.54     495 2442.56  510.16 2446.05   524.4 2456.62
   545.4 2458.55   553.2 2472.08   566.4  2501.7     570 2506.38     621 2554.76
   625.1 2560.89   629.3 2572.12   633.5 2579.22   654.5 2596.29   700.7 2629.47
   734.3 2648.67   742.7 2659.76   784.7 2679.65   893.8 2739.22     910 2751.78
#Mann= 3 ,0,0
       0      .1       0   399.3    .035       0  510.16      .1       0
Bank Sta=399.3,510.16
XS Rating Curve= 0 ,0
Exp/Cntr=0.3,0.1

Type RM Length L Ch R = 1 ,269586  ,510.8,500.8,492.7
XS GIS Cut Line= 2
     2282984.553      514445.055     2282095.083      514637.274
#Sta/Elev= 30
       0 2554.12    41.3 2550.86      70  2545.9   143.6 2530.02   180.4 2517.06
   237.7 2489.77   265.7 2480.29   303.3 2471.69   331.9 2452.22   356.4 2449.97
   377.3 2445.08   393.3 2441.91   503.7 2441.91     516 2444.97   532.4 2454.93
   548.8 2457.09   552.9 2459.98   569.2 2477.83   581.5  2487.8   593.8 2500.49
   616.4 2514.18   663.4 2551.53   683.8  2575.7   717.2 2594.04   757.3 2623.35
   794.3 2647.55   802.5 2655.59   818.9  2667.8   863.9 2695.72     910 2728.45
#Mann= 4 ,-1,0
       0     .06       0      70      .1       0   377.3    .035       0
     516      .1       0
Bank Sta=377.3,516
XS Rating Curve= 0 ,0
Exp/Cntr=0.3,0.1

Type RM Length L Ch R = 1 ,269085  ,548.5,535.4,521.9
XS GIS Cut Line= 2
     2282814.035      513926.678     2281947.994      514206.439
#Sta/Elev= 30
       0 2544.12    18.8 2539.05    39.8 2535.58      65 2533.07     121 2531.02
   170.1 2524.29   203.6 2512.15   257.6 2484.84   295.8 2471.35   321.4  2450.2
   327.5  2448.8   342.4 2449.02   349.8 2445.53   363.5 2441.23   485.4 2441.25
     498 2445.75   510.6 2453.72     519 2455.28   531.6 2454.77   624.1 2512.35
   682.9  2551.9   694.5 2562.19   703.9 2579.94   708.1 2584.96   733.4 2607.83
   796.4 2656.91   804.8 2665.85   821.6 2680.09   859.5 2706.92   910.1 2740.36
#Mann= 5 ,-1,0
       0     .06       0     200      .1       0     300     .12       0
   349.8    .035       0     498      .1       0
Bank Sta=349.8,498
XS Rating Curve= 0 ,0
Exp/Cntr=0.3,0.1

Type RM Length L Ch R = 1 ,268550  ,483.9,462.9,447
XS GIS Cut Line= 2
2282682.75444218 513306.829743912281798.44385955513824.025355338
#Sta/Elev= 30
       0 2559.28    67.9 2547.82   105.9 2538.99   155.6  2533.2   167.3 2528.13
   179.1 2527.64   190.7  2521.4   211.2 2514.39   257.9 2517.72   289.9 2507.45
   308.8 2498.08   336.6 2492.53   351.5 2481.71   364.4  2469.3   404.2 2440.95
   410.8 2439.19   475.6 2439.08   509.4  2441.1   570.8 2442.67     583 2445.95
   628.6 2449.13   654.3  2454.2   684.2 2454.19   693.4 2459.77   725.7 2464.59
   795.4 2489.14   929.8 2527.02   965.6 2539.46  1012.3 2559.34  1024.4 2562.45
#Mann= 5 ,-1,0
       0      .1       0      70     .06       0     300      .1       0
   404.2    .035       0   509.4      .1       0
Bank Sta=404.2,509.4
XS Rating Curve= 0 ,0
Exp/Cntr=0.3,0.1

Type RM Length L Ch R = 1 ,268087  ,505.5,500,499.9
BEGIN DESCRIPTION:
channel burned 0.73' for transition from approximate to detailed reach:
lidar = 2438.6
interpolated = 2437.87
END DESCRIPTION:
XS GIS Cut Line= 2
     2282259.937      512904.929     2281621.779      513553.662
#Sta/Elev= 30
       0 2536.09    48.1 2524.26   107.5 2506.62   121.6 2505.99   152.7 2500.74
   219.2 2491.03   248.9 2483.17     280 2480.21   305.5 2477.78   320.2  2478.1
   331.4  2476.4   347.6 2468.65   365.1 2454.21   375.6 2442.08   381.8 2437.87
   490.2 2437.89   505.3 2441.97   514.8 2445.81   530.1 2448.29   543.1 2453.08
   581.5 2454.85   611.9 2488.54   622.3 2498.72   664.7 2531.77   730.4 2589.66
   806.1 2642.69   815.3 2652.48   838.1 2670.58   875.7 2696.07     910 2716.83
#Mann= 7 ,-1,0
       0      .1       0    48.1     .06       0   152.7      .1       0
     280     .12       0   320.2    .025       0   375.6    .035       0
   505.3      .1       0
Bank Sta=375.6,505.3
XS Rating Curve= 0 ,0
Exp/Cntr=0.3,0.1

Type RM Length L Ch R = 1 ,267587  ,502.7,500,503.8
BEGIN DESCRIPTION:
channel burned 1.43' for transition from approximate to detailed reach:
lidar = 2438
interpolated = 2436.57
c/e of 0.5/0.7 used to correct drawdown
END DESCRIPTION:
XS GIS Cut Line= 2
     2281911.376      512543.247     2281276.822      513195.506
#Sta/Elev= 30
       0  2468.8    20.6 2464.49    69.7 2461.16   130.8 2452.43   153.7 2446.28
   181.3 2448.53     198 2448.02   221.4 2442.33   231.5 2442.44   241.2 2444.37
   251.3 2441.77   285.7 2439.71   315.2 2441.57   362.9 2440.06   383.2 2443.59
   394.7 2440.91   405.3 2436.58   486.4 2436.57   497.9 2440.94   510.5 2451.19
   515.1 2453.61   543.9 2453.75   549.6 2454.97   555.3 2459.42   569.4 2473.84
   623.1 2509.71   702.3 2569.77   778.7 2616.78   795.1 2630.01     910 2693.11
#Mann= 4 ,-1,0
       0     .06       0   251.3      .1       0   394.7    .035       0
   497.9      .1       0
Bank Sta=394.7,497.9
XS Rating Curve= 0 ,0
Exp/Cntr=0.7,0.5

Type RM Length L Ch R = 1 ,267087  ,345.1,433.1,462.1
BEGIN DESCRIPTION:
channel burned 1.76' for transition from approximate to detailed reach:
lidar = 2437.03
interpolated = 2435.27
END DESCRIPTION:
XS GIS Cut Line= 2
     2281559.954      512210.729      2280902.69      512840.097
#Sta/Elev= 30
       0 2461.28    24.2 2443.91    32.5 2441.92      44 2441.65    55.3 2437.97
    89.3 2436.94   131.7 2440.14   160.3 2440.48     188 2440.54     259 2446.42
   304.3 2447.84   362.1 2443.65     375 2443.95   389.2 2438.32   398.4 2435.27
   506.7 2435.32   513.6 2438.12   522.1 2441.79   533.4 2450.58   539.1 2453.25
   575.7 2454.75   587.2 2462.99   601.3 2477.48   610.8  2484.3   657.9 2501.89
   738.1 2528.13   785.2 2547.13   842.2 2567.26   865.3 2577.46     910 2600.04
#Mann= 5 ,-1,0
       0     .06       0    32.5      .1       0   160.3     .05       0
   389.2    .035       0   513.6      .1       0
Bank Sta=389.2,513.6
XS Rating Curve= 0 ,0
Exp/Cntr=0.3,0.1

Type RM Length L Ch R = 1 ,266654  ,128.5,170.4,208.4
BEGIN DESCRIPTION:
channel burned 1.44' for transition from approximate to detailed reach:
lidar = 2435.59
interpolated = 2434.15
END DESCRIPTION:
XS GIS Cut Line= 3
2281538.13606601511904.7040496242280787.98099602512268.923028797
2280669.19187594512495.782549398
#Sta/Elev= 30
       0 2566.74    37.8  2545.9    51.1 2534.39    79.6 2522.05     140 2488.25
   157.5 2486.75     180 2473.52   220.1 2457.53   273.4 2435.48     309  2434.8
   322.3 2439.56   335.7 2440.86     367  2440.5   442.4 2445.45   495.9 2445.48
   513.1 2437.54   522.4 2434.15   660.3 2434.31   669.3  2437.3   704.7  2442.9
   718.1 2440.43   761.2 2440.88   784.8 2450.85   802.6 2453.96   836.9 2455.34
   860.6 2472.84   928.8 2499.48  1023.2 2550.09  1066.3 2575.51    1090 2584.58
#Mann= 7 ,-1,0
       0      .1       0    51.1     .06       0   220.1      .1       0
   273.4     .05       0   442.4    .025       0   513.1    .035       0
   669.3      .1       0
Bank Sta=513.1,669.3
XS Rating Curve= 0 ,0
Exp/Cntr=0.3,0.1

Type RM Length L Ch R = 1 ,266483  ,357,318.7,252.2
BEGIN DESCRIPTION:
start of GRM detailed reach - channel burned 0.64:
lidar invert = 2434.34
effective invert = 2433.70
END DESCRIPTION:
XS GIS Cut Line= 5
2281419.10636355511762.4417602272281121.03407848511975.911614425
2280943.49937513512005.227035806 2280761.8645678512036.079336315
2280517.74235263 512340.89434348
#Sta/Elev= 30
       0 2615.95    81.5 2559.78   118.7 2530.25   141.4 2519.88     166 2500.03
   175.8  2499.2   282.1 2436.18   322.3 2435.74   333.2 2439.78   428.3 2442.01
   436.4 2441.92   448.1 2437.27   460.7  2433.8   570.2  2433.7   586.5 2437.08
     627 2442.04   663.5 2439.11   752.7 2439.75   775.5 2442.65   798.2 2450.97
   812.5 2452.94     845 2453.13   901.3 2450.41   937.7 2453.76   952.6 2459.39
   967.9 2476.38   983.3 2483.11  1037.3 2493.39  1094.2 2492.97  1121.3 2488.47
#Mann= 9 ,-1,0
       0      .1       0     166    .016       0   175.8      .1       0
   282.1     .04       0   322.3     .06       0   448.1    .035       0
   586.5     .08       0   812.5    .016       0     845      .1       0
Bank Sta=448.1,586.5
XS Rating Curve= 0 ,0
Exp/Cntr(USF)=0,0
Minor Loss Coefficient=0
Exp/Cntr=0.3,0.1

Type RM Length L Ch R = 1 ,266165  ,216.2,205.2,173.7
BEGIN DESCRIPTION:
channel burned 0.11':
lidar invert = 2431.80
interpolated invert = 2431.69
END DESCRIPTION:
XS GIS Cut Line= 3
2281169.43474417511526.9809437362280560.87049225511887.789788751
2280329.95283144511933.492242453
#Sta/Elev= 30
       0 2604.54    52.2 2577.71    89.8 2550.26   101.8 2545.57   116.4 2535.75
   133.9 2522.43   142.7 2513.14   148.5  2507.3   164.2 2504.92   187.5 2480.76
   192.5 2473.21   215.6  2451.5   238.6 2434.75   253.6 2431.69   355.8 2431.88
   387.4 2434.63     406 2444.16   480.4 2444.36   591.3 2443.92   600.4 2445.54
   647.7  2445.9   719.5 2452.78   785.7 2454.17   797.9 2458.83   810.1 2459.83
   817.7 2464.33   826.4 2470.61   867.2 2488.67   916.9 2516.17   942.9 2527.12
#Mann= 9 ,-1,0
       0      .1       0   142.7     .06       0   238.6    .035       0
   387.4      .1       0   480.4     .07       0   591.3      .1       0
   600.4     .07       0   719.5     .05       0   817.7      .1       0
Bank Sta=238.6,387.4
XS Rating Curve= 0 ,0
Exp/Cntr(USF)=0,0
Exp/Cntr=0.3,0.1

Type RM Length L Ch R = 1 ,265960  ,221.7,227.6,241.4
BEGIN DESCRIPTION:
channel burned 0.45':
lidar invert = 2430.85
effective invert = 2430.40
END DESCRIPTION:
XS GIS Cut Line= 2
2281032.69923572511312.6698967672280301.86955383511921.324103233
#Sta/Elev= 30
       0 2633.63    29.1 2618.14    82.1 2582.04   111.5 2557.08   122.9 2551.18
   151.3 2527.19   176.8 2500.24   186.9 2499.43   193.9 2495.34   205.2 2483.35
   229.7 2463.59   242.1 2444.13   253.5 2434.09   266.2 2430.47   363.3  2430.4
   378.5 2433.58     387 2437.62   406.7 2440.45     490 2439.65   500.4 2441.32
   588.9 2442.09   663.3 2446.99   682.4 2446.11   700.8 2452.63   710.8 2452.88
   771.1 2454.86   797.1    2470   844.3 2486.25   901.2 2518.48   951.1 2539.26
#Mann= 9 ,-1,0
       0      .1       0   176.8    .016       0   186.9      .1       0
   253.5    .035       0   378.5     .05       0     490     .08       0
   500.4     .05       0   700.8    .016       0   710.8      .1       0
#Block Obstruct= 2 ,-1
   455.4  530.72 2460.22  545.88  622.55  2463.9
Bank Sta=253.5,378.5
XS Rating Curve= 0 ,0
Exp/Cntr=0.7,0.5

Type RM Length L Ch R = 1 ,265732  ,220.6,219.6,217
BEGIN DESCRIPTION:
channel burned 0.83':
lidar invert = 2430.62
interpolated invert = 2429.79
END DESCRIPTION:
XS GIS Cut Line= 2
2280842.30139136511199.8475909222280226.52096253 511637.62898954
#Sta/Elev= 30
       0 2564.35     8.2 2561.73    74.2 2522.04    95.9 2506.99   110.6 2492.19
   114.4 2490.44     123  2489.4   126.6 2487.24   148.8 2467.06   161.1 2444.26
   181.8 2432.83   188.7    2430     194 2429.79   292.2  2429.8     302 2432.84
   311.8 2437.12   326.6 2438.72   351.1 2437.41   360.9 2437.18   381.1 2439.49
   424.7 2437.17   485.5 2438.43   515.9 2444.69   590.5  2448.4   622.1 2451.02
   651.2 2451.01   660.3 2452.74   678.8 2461.24   714.2 2483.45   755.5 2503.42
#Mann= 6 ,-1,0
       0      .1       0   110.6     .06       0   181.8    .035       0
     302    .025       0   351.1     .05       0   590.5      .1       0
Bank Sta=181.8,302
XS Rating Curve= 0 ,0
Exp/Cntr(USF)=0,0
Exp/Cntr=0.3,0.1

Type RM Length L Ch R = 1 ,265513  ,167.1,167.3,168.2
BEGIN DESCRIPTION:
channel burned 1.14':
lidar invert = 2430.34
effective invert = 2429.20
END DESCRIPTION:
Node Name=W
XS GIS Cut Line= 2
2280746.74635135510994.9053429322280073.13952902511485.595442181
#Sta/Elev= 30
       0 2566.42     6.3 2564.26    24.2 2552.56    52.1 2538.59    92.3 2526.63
   112.1  2518.3   132.3 2507.69   156.6 2492.08   166.9 2480.43   172.4  2476.6
   183.6 2475.97   189.6 2474.41  242.62 2432.83   250.6  2429.2   357.1 2429.28
   369.4 2432.64   379.3 2435.44   394.1 2436.42   418.9 2437.59   468.4 2436.38
   513.1 2439.83   588.1 2441.59   626.7 2444.02   639.1 2447.78   666.3 2449.62
     701 2449.13   715.8  2455.4   744.4  2473.7   759.3 2485.48   833.4 2531.62
#Mann= 9 ,-1,0
       0      .1       0   112.1     .06       0   172.4    .016       0
   183.6      .1       0  242.62    .035       0   369.4     .08       0
   394.1     .05       0   639.1    .016       0   666.3      .1       0
Bank Sta=242.62,369.4
XS Rating Curve= 0 ,0
Exp/Cntr=0.3,0.1

Type RM Length L Ch R = 1 ,265345  ,176.9,173,164.6
BEGIN DESCRIPTION:
channel burned 1.34':
lidar invert = 2430.16
interpolated invert = 2428.82
END DESCRIPTION:
XS GIS Cut Line= 2
2280633.03226125510872.7142381082280005.22487092511324.927990527
#Sta/Elev= 30
       0 2570.99    30.6 2551.31    65.1 2531.93    89.8 2520.13   121.3 2501.18
   164.3 2471.46   173.6 2461.83   178.5 2460.28   188.4 2459.57   198.7 2451.59
     213 2443.77   221.6 2436.03   232.8 2432.41   242.6 2428.82     356 2428.84
   367.7 2432.27   384.9 2435.61     460 2436.85   486.7 2438.02   505.3 2437.03
   568.8 2440.07   582.5 2441.85   612.3 2446.84     637 2448.25   677.2 2447.77
   691.2 2453.59   710.9 2465.32   728.8 2474.04   739.9  2480.6   773.7 2494.92
#Mann= 7 ,-1,0
       0      .1       0   121.3     .06       0   221.6     .08       0
   232.8    .035       0   367.7     .05       0     460     .06       0
   582.5      .1       0
Bank Sta=232.8,367.7
XS Rating Curve= 0 ,0
Exp/Cntr(USF)=0,0
Exp/Cntr=0.7,0.5

Type RM Length L Ch R = 1 ,265172  ,278.7,283.6,293.9
BEGIN DESCRIPTION:
channel burned 1.51':
lidar invert = 2429.94
interpolated invert = 2428.43
END DESCRIPTION:
XS GIS Cut Line= 2
2280545.96359794510701.9713194952279788.63565133511308.551523177
#Sta/Elev= 30
       0  2592.4    12.5 2581.45    22.8 2578.54    27.9  2575.5   157.2 2484.22
   171.5 2474.84   211.3 2453.38   222.6 2444.71   236.9 2444.34   256.8 2431.98
   262.5 2428.66   268.2 2428.43   391.8 2428.44   396.9 2431.78     402 2434.48
   413.3 2435.59   622.4 2439.29   660.9  2446.7     689 2446.81   703.6 2446.19
   719.8 2450.99   740.6 2460.23   754.8 2462.31   817.7 2493.74   828.8 2497.74
     843 2506.01   904.3  2525.2   924.8 2528.08   945.5 2534.19   970.3 2543.74
#Mann= 8 ,-1,0
       0      .1       0   222.6    .016       0   236.9      .1       0
   256.8    .035       0   396.9     .05       0   413.3    .016       0
   622.4     .05       0     689      .1       0
Bank Sta=256.8,396.9
XS Rating Curve= 0 ,0
Exp/Cntr(USF)=0,0
Exp/Cntr=0.3,0.1

Type RM Length L Ch R = 1 ,264889  ,331.6,302.4,271.8
BEGIN DESCRIPTION:
channel burned 1.79':
lidar invert = 2429.59
effective invert = 2427.80
END DESCRIPTION:
XS GIS Cut Line= 3
2280376.79984316510499.0798719552279722.24897383510959.067224495
 2279643.2494382511129.774570226
#Sta/Elev= 30
       0 2555.55    42.2 2525.41    64.3 2512.25   113.2 2487.67   122.5 2480.76
   142.8 2469.48   154.1  2461.7     167 2450.06   177.6 2448.15   188.6 2441.02
   205.8 2437.49   225.7 2436.95   245.2 2430.93   254.1 2427.82   377.2  2427.8
   388.7 2431.06   421.1 2434.47   599.2 2437.14   641.2 2444.65   713.2 2444.23
   741.1  2446.4     755 2448.39   818.2 2473.88   854.4 2481.99   881.1 2494.37
   894.9 2498.41   930.2 2504.36   947.8 2505.69   965.4 2509.51   988.1 2510.75
#Mann= 9 ,-1,0
       0      .1       0   205.8    .016       0   225.7      .1       0
   245.2    .035       0   388.7     .05       0   421.1    .016       0
   599.2     .06       0   741.1     .08       0   894.9      .1       0
Bank Sta=245.2,388.7
XS Rating Curve= 0 ,0
Exp/Cntr=0.3,0.1

Type RM Length L Ch R = 1 ,264586  ,253.4,196.8,179.9
BEGIN DESCRIPTION:
structure xs 4 - channel burned 1.91':
lidar invert = 2428.32
interpolated invert = 2426.41
END DESCRIPTION:
XS GIS Cut Line= 4
2280235.80065629510185.2345462982280060.44755762510308.631171293
2279854.78651596510529.446184442   2279547.37738510826.031055044
#Sta/Elev= 30
       0 2570.54     4.4 2568.59    42.8 2542.24    77.2 2517.48   120.3 2490.77
   186.3 2453.31   212.1  2441.7   234.8 2436.21   277.3 2436.05   291.7 2435.28
   308.1 2431.22  312.48 2429.04     319 2426.41   438.6  2426.5  447.78 2429.02
   475.4 2430.04   499.4 2433.69   547.6 2434.53   636.5 2436.15   673.4 2436.14
   714.3 2443.23   758.8 2443.53   778.1  2442.3   792.2 2442.29   817.7 2449.41
   826.2 2450.04   832.6 2450.66   855.7  2458.8   907.5 2484.25   943.3 2502.02
#Mann= 11 ,-1,0
       0      .1       0   120.3     .06       0   212.1     .08       0
   277.3     .07       0  312.48    .035       0  447.78     .08       0
   547.6      .1       0   636.5     .08       0   778.1     .07       0
   826.2     .06       0   907.5      .1       0
#Block Obstruct= 1 ,-1
  796.03  845.18 2473.72
Bank Sta=312.48,447.78
XS Rating Curve= 0 ,0
Exp/Cntr(USF)=0,0
Exp/Cntr=0.5,0.3

Type RM Length L Ch R = 1 ,264389  ,142.4,93,90.9
BEGIN DESCRIPTION:
structure xs 3
channel burned per surveyed cross section points
END DESCRIPTION:
XS GIS Cut Line= 6
2279683.51081002509503.9175108352279689.23320511 509687.03415369
2279768.03512668509865.0191509642279883.70540758510019.246192167
 2279898.1641927510096.3597127682279492.42493398510795.754165263
#Sta/Elev= 30
       0 2468.25    37.3 2459.04    73.3  2455.7   125.3 2446.07   141.1 2440.69
   161.3 2439.84   241.2  2439.8   288.4  2427.7   392.7 2430.63   658.6  2433.9
   690.5 2435.83   700.3 2436.19   791.5 2435.99  827.76 2427.09  841.53 2424.57
  917.44 2424.44   936.9 2426.02    1026 2435.19  1082.2 2437.23  1096.3 2440.16
  1135.7 2437.64  1194.8  2442.6  1260.8 2443.63  1275.4 2450.99  1327.7 2454.08
  1344.8 2463.55  1358.9 2468.25  1400.5 2482.59    1447 2501.84  1460.4 2503.69
#Mann= 14 ,-1,0
       0      .1       0   161.3     .06       0   392.7     .08       0
   690.5    .016       0   700.3     .06       0  827.76    .035       0
   936.9     .08       0    1026    .016       0  1082.2     .06       0
  1096.3    .016       0  1135.7     .06       0  1194.8    .016       0
  1260.8     .06       0  1358.9      .1       0
#XS Ineff= 3 ,-1
       0     792  2431.5    1022 1103.32  2439.9 1103.32 1311.55    2445
Permanent Ineff=
       F       F       F
#Block Obstruct= 2 ,-1
  1204.6 1243.17 2463.46  1281.7 1330.98 2475.09
Bank Sta=827.76,936.9
XS Rating Curve= 0 ,0
Exp/Cntr=0.5,0.3

Type RM Length L Ch R = 3 ,264345  ,,,
BEGIN DESCRIPTION:
Bridge No.: 54075GRM010 Cass Rd (Route 66)
JV notes: road deck updated per surveyed XS data points
channel burned per surveyed cross sections
structure opening based on survey data, photos, and aerial imagery
surveyed inverts are 2-3' below inverts from lidar:
 surveyed invert US is 2424.75
 surveyed invert DS is 2422.27
END DESCRIPTION:
Bridge Culvert--1,0,-1,-1, 0
Deck Dist Width WeirC Skew NumUp NumDn MinLoCord MaxHiCord MaxSubmerge Is_Ogee
27,40,2.6,0, 411, 411, , , 0.98, 0, 0,0,,
      34    36.4    40.4    44.4    45.1    47.6    48.4    49.3    51.5    52.4
    56.4    57.6    59.2    60.4    61.8      63    64.4    68.4    72.4    74.3
    78.4    80.4    82.2    82.7    84.4    88.4    89.9    92.4    96.4    97.6
   100.5   104.5   107.8   109.1   111.9   112.5   116.5   120.5   120.6   124.5
   132.8     136   139.9   140.5   141.2   143.7   145.4   147.5   148.5   149.5
   151.4   152.5   153.7   155.2   156.5   157.9   159.1   162.1   162.9   164.5
   166.2   166.8   168.5   172.5   176.5   180.5   188.5   196.5   208.6   210.9
   213.3   216.9   221.1   222.9   226.1   229.4   233.6   237.8     242   247.7
   248.5   251.8   254.5   259.7   261.4   267.1   267.8   271.7   277.7   279.6
   283.8   297.7   304.7   309.5   317.2   319.1   321.4   325.3   328.6   331.7
   332.6   334.1   336.7   341.1   344.2   346.2   348.1   350.4   351.2   359.9
   362.8   365.9     369     371   372.6   376.8   381.5   384.2   385.9   390.4
     395     396     399   402.5   404.3   405.4   407.6   410.5   413.9   416.3
   418.7     420   422.1   427.4   433.7   436.5   437.7   442.5   445.2   448.1
     451   453.9   457.1   459.7   461.6     464   465.5   468.3   474.1   475.9
     477   480.1   480.7   482.8   485.9   488.4   491.3   491.6     497   501.4
   504.2   506.6   511.7     514   516.9   519.7     522   525.4   527.2   532.4
   535.9   542.2   545.3   547.8   548.5     551     553   558.2   562.4   567.5
   570.9   573.8   579.4   582.3   585.5   588.6   591.1   596.1   597.1   599.3
   601.8   605.9   606.8   609.8   614.1   615.2   623.4   626.4   626.7   630.6
   634.7   636.8   643.4   646.8   650.9   654.9   658.9   660.8   663.4   665.9
   666.9   671.1   673.8   677.3   680.8   681.9   687.7   692.9   697.5   699.9
   700.6   703.6   704.3   706.7   709.7   713.2   717.2     722   725.1   727.9
   728.3   732.2     735   743.5  787.82  814.65  818.74  818.74  867.58  892.28
  906.26  907.38   944.4  995.66  995.66  997.57 1018.33 1062.78  1070.1    1073
  1073.5    1076  1078.9  1081.8  1086.4  1087.4    1092  1099.4  1102.3  1105.2
  1108.1    1111  1111.8  1115.2  1119.7  1119.9  1122.7  1124.5  1125.7  1127.6
  1129.1  1131.5  1133.8  1135.5  1138.4  1140.3  1143.4  1147.7    1149  1151.4
    1152  1153.7  1154.9  1159.3  1160.7  1163.7  1166.2  1167.2  1170.9  1172.4
  1175.3  1178.3  1180.1  1181.2  1184.1    1187  1187.3  1190.9  1192.9  1194.1
  1198.5  1204.6    1208  1210.4  1212.6  1216.3  1219.2  1221.9    1225  1226.5
  1230.4  1232.2  1235.8  1236.7  1238.3  1239.7  1240.4  1243.4  1245.1  1245.5
  1246.3  1248.4  1251.3  1254.2  1257.2    1259    1263  1263.6  1268.2  1268.9
    1270  1272.9  1277.7  1282.2  1285.8  1289.3  1296.1  1299.4  1300.7    1304
  1305.3  1309.8  1314.6  1315.7  1319.3  1321.8  1323.9  1327.3  1328.5    1333
  1336.1  1337.8  1341.2    1342  1342.4  1344.3  1344.9  1347.1  1347.8  1350.7
  1351.7  1356.3    1357  1359.5    1361  1362.4  1364.9  1365.3  1366.7  1370.3
  1371.2  1374.9  1377.9  1379.5    1380  1382.9  1384.2  1388.6  1391.7  1393.4
  1394.6  1396.5  1398.1  1400.4  1402.7  1403.3  1404.4  1409.2  1411.5    1412
  1412.3    1415  1416.6    1418  1420.2  1421.3  1423.8  1425.9  1426.7  1428.1
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                                                 2435.67 2435.67 2436.02 2436.19
 2436.29  2436.3 2436.56 2436.92 2436.92
     -17   -14.6   -10.6    -6.6    -5.9    -3.4    -2.6    -1.7      .5     1.4
     5.4     6.6     8.2     9.4    10.8      12    13.4    17.4    21.4    23.3
    27.4    29.4    31.2    31.7    33.4    37.4    38.9    41.4    45.4    46.6
    49.5    53.5    56.8    58.1    60.9    61.5    65.5    69.5    69.6    73.5
    81.8      85    88.9    89.5    90.2    92.7    94.4    96.5    97.5    98.5
   100.4   101.5   102.7   104.2   105.5   106.9   108.1   111.1   111.9   113.5
   115.2   115.8   117.5   121.5   125.5   129.5   137.5   145.5   157.6   159.9
   162.3   165.9   170.1   171.9   175.1   178.4   182.6   186.8     191   196.7
   197.5   200.8   203.5   208.7   210.4   216.1   216.8   220.7   226.7   228.6
   232.8   246.7   253.7   258.5   266.2   268.1   270.4   274.3   277.6   280.7
   281.6   283.1   285.7   290.1   293.2   295.2   297.1   299.4   300.2   308.9
   311.8   314.9     318     320   321.6   325.8   330.5   333.2   334.9   339.4
     344     345     348   351.5   353.3   354.4   356.6   359.5   362.9   365.3
   367.7     369   371.1   376.4   382.7   385.5   386.7   391.5   394.2   397.1
     400   402.9   406.1   408.7   410.6     413   414.5   417.3   423.1   424.9
     426   429.1   429.7   431.8   434.9   437.4   440.3   440.6     446   450.4
   453.2   455.6   460.7     463   465.9   468.7     471   474.4   476.2   481.4
   484.9   491.2   494.3   496.8   497.5     500     502   507.2   511.4   516.5
   519.9   522.8   528.4   531.3   534.5   537.6   540.1   545.1   546.1   548.3
   550.8   554.9   555.8   558.8   563.1   564.2   572.4   575.4   575.7   579.6
   583.7   585.8   592.4   595.8   599.9   603.9   607.9   609.8   612.4   614.9
   615.9   620.1   622.8   626.3   629.8   630.9   636.7   641.9   646.5   648.9
   649.6   652.6   653.3   655.7   658.7   662.2   666.2     671   674.1   676.9
   677.3   681.2     684   692.5  736.82  763.65  767.74  767.74  816.58  841.28
  855.26  856.38   893.4  944.66  944.66  946.57  967.33 1011.78  1019.1    1022
  1022.5    1025  1027.9  1030.8  1035.4  1036.4    1041  1048.4  1051.3  1054.2
  1057.1    1060  1060.8  1064.2  1068.7  1068.9  1071.7  1073.5  1074.7  1076.6
  1078.1  1080.5  1082.8  1084.5  1087.4  1089.3  1092.4  1096.7    1098  1100.4
    1101  1102.7  1103.9  1108.3  1109.7  1112.7  1115.2  1116.2  1119.9  1121.4
  1124.3  1127.3  1129.1  1130.2  1133.1    1136  1136.3  1139.9  1141.9  1143.1
  1147.5  1153.6    1157  1159.4  1161.6  1165.3  1168.2  1170.9    1174  1175.5
  1179.4  1181.2  1184.8  1185.7  1187.3  1188.7  1189.4  1192.4  1194.1  1194.5
  1195.3  1197.4  1200.3  1203.2  1206.2    1208    1212  1212.6  1217.2  1217.9
    1219  1221.9  1226.7  1231.2  1234.8  1238.3  1245.1  1248.4  1249.7    1253
  1254.3  1258.8  1263.6  1264.7  1268.3  1270.8  1272.9  1276.3  1277.5    1282
  1285.1  1286.8  1290.2    1291  1291.4  1293.3  1293.9  1296.1  1296.8  1299.7
  1300.7  1305.3    1306  1308.5    1310  1311.4  1313.9  1314.3  1315.7  1319.3
  1320.2  1323.9  1326.9  1328.5    1329  1331.9  1333.2  1337.6  1340.7  1342.4
  1343.6  1345.5  1347.1  1349.4  1351.7  1352.3  1353.4  1358.2  1360.5    1361
  1361.3    1364  1365.6    1367  1369.2  1370.3  1372.8  1374.9  1375.7  1377.1
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                                                 2435.67 2435.67 2436.02 2436.19
 2436.29  2436.3 2436.56 2436.92 2436.92
Pier Skew, UpSta & Num, DnSta & Num=  ,897.38, 2 ,848.56, 2 , 0 , 0 , 0 ,,
       3       3
       0    2437
       3       3
       0    2437
BR Coef=-1 ,-1 , 0 ,, 0 ,,,0.8,0,1.33,0,
WSPro=,,,, 1 ,,,, 0 ,,,, 0 ,,,,-1 ,-1 ,-1 , 0 , 0 , 0 , 0 , 0
BR U #Sta/Elev= 414
       0 2468.25     1.9 2467.75     4.7 2466.62     8.9 2465.54    17.3 2463.91
    21.3 2463.03    25.4 2462.06    32.9 2459.85    37.3 2459.04    41.9 2458.48
    45.3  2458.2    53.3 2457.74    61.3 2456.81    69.3 2456.28    73.3  2455.7
    77.3  2455.1    89.3 2452.84    93.3 2451.94   109.3 2448.65   113.3 2447.95
   117.3 2447.09   125.3 2446.07   129.3 2445.16   132.8 2443.77   136.9 2442.03
   141.1 2440.69   145.2 2440.06   149.3 2439.84   161.3 2439.84   173.3 2440.26
   178.3 2440.18     184 2439.86   187.1 2439.85   191.4 2439.98   196.4 2439.85
   202.7 2439.91   208.8 2439.82   215.5 2439.97   219.8 2439.92   224.7 2440.11
   232.7 2440.22   233.5 2440.14     237 2440.02   239.7 2439.82   241.2  2439.8
   242.8 2439.55   244.7 2439.36   245.5 2439.25     249  2438.5   254.1 2437.51
   258.3 2436.46   262.7 2434.62     267 2432.94   267.6 2432.74   271.3  2431.2
   273.8  2430.5   275.5 2429.93   276.9 2429.67   279.9 2428.84     283  2428.4
   284.1 2428.07   288.4  2427.7   292.3 2427.72     297 2427.61   301.3 2427.69
   307.5 2428.03   310.5 2428.03   316.4 2428.44   319.3 2428.52   322.3 2428.88
   323.9 2428.98   328.5 2428.97   331.2 2429.09   337.1 2429.25   346.6 2429.46
   351.2 2429.64   351.8 2429.67   355.7 2429.96   360.2 2430.14   373.9 2430.27
   383.4 2430.55   392.7 2430.63   412.7 2430.98   429.9 2431.11   431.8 2431.17
   433.4  2431.2   445.1 2431.34   458.3 2431.62   458.4 2431.62   461.3 2431.59
   463.4 2431.56   465.1 2431.54   478.3 2431.69   493.4 2431.66   505.1 2431.77
   512.7 2431.75   524.1    2432   538.4 2432.09   555.6 2432.57   572.8 2433.24
   587.9 2433.43   601.4 2433.51   612.9 2433.77   621.8 2433.84   638.1 2434.15
   646.2 2434.12     648 2434.08   651.7 2433.96   653.6 2433.92   654.5  2433.9
     655 2433.89   658.6  2433.9   659.4 2433.93   662.8 2434.04   665.2 2434.21
   666.9 2434.33     671 2434.71   690.5 2435.83   700.3 2436.19   708.5 2436.24
     710 2436.16   712.7 2436.02   713.2 2436.02   716.4 2436.02   716.9 2436.01
   719.7 2436.01   735.3 2436.46   737.1 2436.55   739.6 2436.73     740 2436.75
   740.2 2436.76   744.6 2436.91   747.8 2436.98   748.8 2436.98   749.3 2436.98
   751.7 2436.84   751.7 2436.83     754 2436.64   754.6 2436.58   755.5 2436.49
   758.7 2436.32   760.4 2436.14   763.2 2436.05   763.3 2436.04   768.1 2435.81
   769.1 2435.84   770.8  2435.9     772 2435.88   772.8 2435.87   774.9 2435.95
   777.9  2436.1   780.8 2436.24   782.2 2436.27   786.6 2436.17   786.8 2436.16
   787.9 2436.12   789.5 2436.06   791.5 2435.99   796.2 2435.49   801.1 2434.51
   805.6 2432.88   806.9 2432.44   810.3 2431.43   815.7 2430.11  818.67  2429.4
  827.76 2427.09  834.39 2425.36  841.53 2424.57  865.48 2424.76  892.17 2424.75
  907.27 2424.95  917.44 2424.44  924.35 2424.96   936.9 2426.02  953.65 2427.38
  982.13 2429.79   996.1 2432.57   997.8 2432.77     999 2432.91  1000.8 2433.13
  1002.5 2433.33  1004.8 2433.53  1005.2 2433.58  1007.2  2433.8  1007.7 2433.84
  1013.5 2434.14  1016.2 2434.25  1016.4 2434.27  1016.6 2434.28  1017.3 2434.36
  1019.3 2434.59  1021.3 2434.79  1022.2 2434.92  1023.8 2435.05    1026 2435.19
  1028.1 2435.31  1030.7 2435.39    1031  2435.4  1051.3 2435.76  1053.5 2435.82
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BR U #Mann= 14
       0      .1   161.3     .06   392.7     .08   690.5    .016   700.3     .06
  827.76     .03   936.9     .08    1026    .016  1082.2     .06  1096.3    .016
  1135.7     .06  1194.8    .016  1260.8     .06  1358.9      .1
BR D #Sta/Elev= 416
       0 2452.09     3.8 2451.54     7.9 2450.61      11 2449.74    11.7  2449.6
    14.6 2449.19    19.7 2448.64    23.8 2448.01    27.8 2447.23    36.2 2446.31
    44.5 2445.28    51.9 2444.27      56 2443.29      60 2442.03      65  2440.6
    67.3 2440.17    68.6 2439.88    73.5 2439.85      83 2439.94    88.2 2439.92
    92.2 2439.85    96.3 2439.73   104.7  2439.3   108.3 2439.03   111.9  2438.7
   115.5 2438.22   119.1 2437.59   129.9 2435.32   132.5 2434.88   137.1 2434.31
   141.5 2433.99   152.6 2433.55   157.6 2433.48   165.1 2433.61   177.1 2433.46
   181.2 2433.36   185.5 2433.38   189.4 2433.34   193.5 2433.03   195.3 2432.81
     196 2432.77   198.7 2432.47   201.7 2432.05   203.4 2431.93   205.8 2431.69
   208.7 2430.97   212.1 2430.25     214 2429.81   215.4 2429.87   222.1  2429.9
   226.3 2429.97   230.4 2430.24   235.6 2430.44   240.4  2430.7   243.3 2430.79
   245.6 2430.78   250.9 2430.97     255 2430.92   263.2 2430.18   269.1 2429.93
   272.5 2429.83   274.9 2429.87   275.5 2429.86   279.2 2429.56   279.6 2429.55
   282.5 2429.46   283.7 2429.44   285.4 2429.42   287.8 2429.41   289.2 2429.33
   290.7 2429.27   291.8 2429.21     296 2428.81     300 2428.46     306 2428.41
   308.2 2428.46   311.7 2427.84   312.3 2427.73   314.5 2427.56   316.1 2427.43
   324.6 2426.32   326.2 2426.19   328.7 2425.99   332.7 2426.09   332.8  2426.1
   332.9 2426.11   333.1 2426.16   334.2 2426.43     336 2426.76   337.2 2426.87
   338.9 2427.28   341.8  2427.8   346.4 2428.51   350.2 2428.89     351 2428.99
   353.6 2429.36   358.4 2429.72   360.1 2429.83   362.3 2429.86   362.4 2429.87
   365.4 2429.91   366.6 2430.01   369.3 2430.18   371.3 2430.36   373.8 2430.69
   374.2 2430.71   377.1 2430.98   378.4 2431.18   380.1 2431.31   382.8 2431.55
     383 2431.56   394.8  2431.8   410.4 2431.96   432.5 2431.78   438.7 2431.81
     444 2431.75   454.7 2431.75   455.7 2431.76   456.8 2431.79   458.6 2431.83
   472.7 2431.88   474.9 2431.92   475.6 2431.92   476.1 2431.93   501.1 2431.96
   518.1 2432.15   540.7  2432.2   554.9 2432.36     575 2432.81   575.7 2432.83
   577.1 2432.88   578.2 2432.92   579.9 2432.98   581.4 2433.04     583 2433.09
   584.6 2433.15   586.5 2433.26   587.8 2433.34   588.2 2433.36   588.9 2433.38
   591.1 2433.45   592.2 2433.49   596.4 2433.74   597.7 2433.81   599.1 2433.89
   600.4 2433.97   601.5 2434.04   604.4 2434.22   605.3 2434.28   607.6 2434.46
   608.4 2434.52   612.4 2434.87     616 2434.95   616.4 2434.96   616.8 2434.96
   620.2 2434.95   624.4 2434.94   628.2 2434.78   628.4 2434.77   632.4 2434.65
   632.9 2434.64   637.1  2434.6   663.4 2435.34     668 2435.51   686.3 2436.34
   686.9 2436.37   687.9 2436.42   689.8 2436.51   690.9 2436.57   692.7 2436.66
   694.8 2436.77   695.5 2436.81   695.7 2436.82     696 2436.84   698.6 2436.97
   700.1 2437.05   701.6  2437.1   704.5 2437.18   712.4 2437.36   713.3 2437.38
   713.8 2437.38   715.6 2437.38   718.4 2437.43   719.2 2437.45   722.1 2437.55
     723  2437.6   725.1 2437.69   726.1 2437.73   727.6 2437.79     728  2437.8
   728.8 2437.81   732.2 2437.92   733.9 2437.96   736.5 2437.99   736.7    2438
   741.3 2437.96   742.7 2437.91   745.1 2437.82   745.9 2437.79   746.9 2437.66
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BR D #Mann= 11
       0      .1      83    .016    96.3      .1   410.4    .016   715.6     .06
  786.44     .03  909.71     .07  935.56     .08   979.8    .016  1181.6     .06
  1317.7      .1
BR D Banks=786.44,
BC Design=,, 0 ,, 0 ,,,,,,
BC Use User HTab Curves=0
BC User HTab FreeFlow(D)= 0

Type RM Length L Ch R = 1 ,264296  ,446.4,512,522.2
BEGIN DESCRIPTION:
structure xs 2
channel burned per surveyed cross section points
END DESCRIPTION:
XS GIS Cut Line= 6
2279644.82985845509509.5914973012279626.28685913509666.052038363
2279664.41383337509838.5113782582279789.72330435510012.016799611
2279799.36249443510101.1793078062279442.71246165510737.365852767
#Sta/Elev= 30
       0 2452.09    51.9 2444.27    68.6 2439.88      83 2439.94    96.3 2439.73
   141.5 2433.99   189.4 2433.34     214 2429.81     255 2430.92   328.7 2425.99
   382.8 2431.55   410.4 2431.96   554.9 2432.36   715.6 2437.38   750.5  2437.2
  780.39 2426.82  786.44 2424.94  843.85 2422.27  897.98 2424.28  909.71 2426.39
  931.33 2432.91   979.8 2438.43  1172.4 2446.32  1181.6 2449.97  1190.7 2452.31
  1277.9 2455.57  1282.4 2457.38  1291.6 2467.04  1317.7 2477.03  1369.8 2498.15
#Mann= 11 ,-1,0
       0      .1       0      83    .016       0    96.3      .1       0
   410.4    .016       0   715.6     .06       0  780.39    .035       0
  909.71     .07       0  931.33     .08       0   979.8    .016       0
  1181.6     .06       0  1317.7      .1       0
#XS Ineff= 2 , 0
             759  2431.5   953.3          2439.9
Permanent Ineff=
       F       F
#Block Obstruct= 2 ,-1
  632.38  640.45 2454.69  1194.6 1273.98 2475.43
Bank Sta=780.39,909.71
XS Rating Curve= 0 ,0
Exp/Cntr(USF)=0,0
Exp/Cntr=0.5,0.3

Type RM Length L Ch R = 1 ,263784  ,503.9,473.7,470.2
BEGIN DESCRIPTION:
xs 1 - channel burned 0.66':
lidar invert = 2423.96
effective invert = 2423.30
END DESCRIPTION:
XS GIS Cut Line= 2
2279630.50653587509511.5940303752279059.55465616510284.323919234
#Sta/Elev= 30
       0 2447.19    17.4 2440.92    28.5 2440.12    48.6 2440.32    71.2  2434.1
   134.4 2431.11   178.9 2426.18     206 2429.03   243.1 2425.73   280.5 2429.24
   293.4 2428.67   310.3 2427.39   391.8 2431.12   494.3 2429.07     509  2430.4
   523.3 2426.58   534.8 2423.31   652.1  2423.3   663.6 2423.32   674.9 2426.47
   698.3 2437.43   737.9 2440.87   760.7 2456.49   769.3 2459.88   800.8 2460.61
   807.7 2460.64     852 2462.68   860.8 2465.65   923.8 2466.53   960.8 2468.87
#Mann= 12 ,-1,0
       0      .1       0    28.5    .016       0    48.6      .1       0
   280.5    .016       0   293.4     .08       0   523.3    .035       0
   674.9      .1       0   760.7     .05       0   800.8     .06       0
   807.7    .016       0     852     .05       0   923.8     .07       0
#Block Obstruct= 1 ,-1
  871.45  921.21 2485.81
Bank Sta=523.3,674.9
XS Rating Curve= 0 ,0
Exp/Cntr(USF)=0,0
Exp/Cntr=0.3,0.1

Type RM Length L Ch R = 1 ,263311  ,531.8,533.5,536.6
BEGIN DESCRIPTION:
channel burned 0.21':
lidar invert = 2422.41
effective invert = 2422.20
END DESCRIPTION:
XS GIS Cut Line= 2
2279419.08231368508938.5395002262278654.56597917510063.139520601
#Sta/Elev= 30
       0 2506.96    12.3 2502.04    32.8 2487.28    90.5 2452.93   133.2 2433.87
   159.5 2433.62   182.2 2430.02   261.3 2428.14   443.3 2430.37   467.6 2428.62
     489  2423.6   525.2 2425.62   560.1 2422.74   637.4 2423.04   670.7 2426.66
   825.4  2428.8   844.7    2429   873.8 2428.84  884.73 2424.46   893.2  2422.2
  1009.2 2422.22  1020.4 2424.41  1038.3 2428.59    1106 2427.26  1130.2 2435.98
  1141.3 2437.35  1155.7 2437.28  1204.7 2454.24  1231.7 2459.34  1359.9 2463.02
#Mann= 13 ,-1,0
       0      .1       0   133.2    .016       0   159.5     .06       0
   467.6      .1       0   525.2     .08       0   825.4    .016       0
   844.7      .1       0  884.73    .035       0  1020.4      .1       0
  1130.2     .07       0  1141.3    .016       0  1155.7     .08       0
  1204.7     .06       0
#Block Obstruct= 3 ,-1
  296.46   350.9 2448.45 1233.04 1262.41 2480.68  1358.3 1359.86 2482.81
Bank Sta=884.73,1020.4
XS Rating Curve= 0 ,0
Exp/Cntr=0.3,0.1

Type RM Length L Ch R = 1 ,262777  ,340.9,575.1,616.7
BEGIN DESCRIPTION:
channel burned 0.14':
lidar invert = 2420.84
effective invert = 2420.70
END DESCRIPTION:
Node Name=V
XS GIS Cut Line= 2
2279057.52665662508574.9175870692278127.44649579509863.058041203
#Sta/Elev= 30
       0 2443.63      16 2433.99    36.5 2434.12    59.9  2429.2   131.5 2427.04
   151.6 2426.88   208.9 2425.65   318.5 2425.92   337.8 2425.91   427.1 2427.75
   589.9  2424.5   637.8 2420.07   706.1 2420.31   753.2 2427.18   772.4 2426.81
   944.7 2427.66   979.4 2422.77  1137.5 2422.64  1152.3 2426.99  1266.1 2428.09
  1280.6 2433.36  1305.3 2435.43  1311.9 2435.87  1349.2 2439.15  1413.8 2453.49
  1469.5 2454.99  1491.9 2461.86  1515.3 2462.54  1535.4 2468.03  1588.8 2470.46
#Mann= 18 ,-1,0
       0      .1       0      16    .016       0    36.5     .06       0
   131.5     .07       0   151.6    .016       0   208.9     .05       0
   318.5    .016       0   337.8     .05       0   589.9      .1       0
   753.2     .07       0   772.4     .05       0   944.7     .08       0
   979.4    .035       0  1137.5      .1       0  1305.3    .016       0
  1311.9     .07       0  1491.9    .016       0  1515.3     .07       0
#XS Ineff= 2 , 0
           332.7 2437.98
Permanent Ineff=
       F       F
#Block Obstruct= 2 ,-1
  493.13  512.41 2446.17  1380.7 1436.72 2473.45
Bank Sta=979.4,1137.5
XS Rating Curve= 0 ,0
Exp/Cntr=0.3,0.1
