HEC-RAS study GRNBRRRV.prj: GRNBRRRV

--- GRNBRRRV.g01 (geometry) --- (continued)

Type RM Length L Ch R = 1 ,262202  ,216.7,359.7,381.7
BEGIN DESCRIPTION:
channel burned 1.35':
lidar invert = 2419.15
effective invert = 2417.80
END DESCRIPTION:
XS GIS Cut Line= 3
2278945.91533007508416.8819300012277798.80092158509211.765371729
2277555.36158263509505.411929548
#Sta/Elev= 30
       0 2439.46    18.7 2439.71    64.7 2428.09     153 2423.58   162.4 2423.44
   291.8 2423.91   306.2 2424.32   440.1 2423.61   459.6 2420.02     518 2421.67
   581.2 2417.98   613.7 2418.95   633.9 2424.53     746 2422.37   941.5 2425.65
  1116.5 2420.49  1125.4 2417.91  1278.7  2417.8  1283.5 2420.62  1292.1 2429.43
  1338.1 2432.78  1349.6  2432.4  1389.1 2433.58  1412.7 2440.44  1537.7 2440.19
  1551.9 2443.92  1580.3 2444.21  1605.3 2446.53  1725.6 2460.46    1777 2472.57
#Mann= 16 ,-1,0
       0    .016       0    18.7     .06       0     153    .016       0
   162.4     .06       0   291.8    .016       0   306.2     .06       0
   440.1     .08       0   633.9      .1       0  1116.5    .035       0
  1283.5     .01       0  1338.1    .016       0  1349.6     .08       0
  1551.9    .016       0  1580.3     .05       0  1605.3      .1       0
  1725.6     .06       0
#XS Ineff= 2 , 0
          380.95 2439.33
Permanent Ineff=
       F       F
#Block Obstruct= 4 ,-1
   56.19  104.04 2447.95  237.35  270.66 2442.05  342.06  374.54 2443.08
 1464.44 1534.16 2458.79
Bank Sta=1116.5,1283.5
XS Rating Curve= 0 ,0
Exp/Cntr=0.3,0.1

Type RM Length L Ch R = 1 ,261842  ,256.1,433.3,458
BEGIN DESCRIPTION:
channel burned 1.86':
lidar invert = 2418.16
interpolated invert = 2416.30
END DESCRIPTION:
XS GIS Cut Line= 3
2278907.73741247508320.338941419 2277577.5291821508867.362978185
2277290.76327737509248.110986154
#Sta/Elev= 30
       0 2444.85    12.5 2444.67    38.5 2437.14     112 2431.46   211.5 2425.09
   254.6 2420.76   354.2 2421.62   384.5 2416.46   548.8 2421.93   868.9 2423.34
   941.2 2418.86   998.6 2422.99  1072.1 2419.96  1089.4  2416.3    1266 2416.41
 1272.25 2420.02  1301.4 2430.41  1312.6 2430.47    1323 2431.89  1331.6 2439.72
  1344.6 2443.67  1450.6 2446.84  1580.5 2454.68    1640 2455.64    1660 2456.31
  1766.1 2462.02  1791.9 2459.62  1826.1 2460.78  1871.9 2471.79    1915 2491.31
#Mann= 15 ,-1,0
       0    .016       0    12.5     .06       0     112    .016       0
   211.5     .06       0   354.2      .1       0  1072.1    .035       0
 1272.25      .1       0  1301.4    .016       0  1312.6     .08       0
  1450.6     .06       0  1580.5      .1       0    1640    .016       0
    1660     .06       0  1791.9    .016       0  1826.1      .1       0
#XS Ineff= 2 , 0
          333.33  2439.8
Permanent Ineff=
       F       F
#Block Obstruct= 3 ,-1
   51.28   89.44 2454.43 1429.94 1438.29 2464.38  1485.1 1510.99 2468.64
Bank Sta=1072.1,1272.25
XS Rating Curve= 0 ,0
Exp/Cntr(USF)=0,0
Exp/Cntr=0.3,0.1

Type RM Length L Ch R = 1 ,261409  ,236,315.2,368.2
BEGIN DESCRIPTION:
channel burned 0.66':
lidar invert = 2415.16
effective invert = 2414.50
END DESCRIPTION:
XS GIS Cut Line= 4
2278638.35199106 508187.186127072278001.82175818508396.265400645
 2277681.2335387 508349.803339852277179.44328212508535.651583028
#Sta/Elev= 30
       0 2434.63   182.1 2433.19     217 2431.89   244.2 2415.95   288.4 2413.91
   310.7 2416.13   390.9  2420.8   486.5 2419.82   561.1 2417.73   659.1 2421.59
   675.7 2417.22   801.3 2415.47   861.3 2420.26     898  2415.7   995.1 2417.64
  1024.9 2424.36  1084.3 2426.04  1131.2 2427.96  1140.1 2428.12  1177.9 2433.47
  1186.5  2434.2  1216.9 2443.85  1233.9 2441.85  1333.5 2442.44  1344.8 2445.87
  1387.5 2445.03  1411.4  2451.6  1420.7 2452.24  1464.3 2469.65    1529 2506.54
#Mann= 16 ,-1,0
       0     .06       0   182.1      .1       0   244.2     .04       0
   310.7      .1       0   486.5     .08       0   675.7    .035       0
   995.1      .1       0  1084.3     .07       0  1131.2    .016       0
  1140.1     .07       0  1177.9    .016       0  1186.5     .05       0
  1233.9     .04       0  1333.5     .05       0  1411.4    .016       0
  1420.7      .1       0
#Block Obstruct= 1 ,-1
  126.73  177.52 2452.55
Bank Sta=675.7,995.1
XS Rating Curve= 0 ,0
Exp/Cntr(USF)=0,0
Exp/Cntr=0.3,0.1

Type RM Length L Ch R = 1 ,261094  ,547,525.4,318.1
BEGIN DESCRIPTION:
channel burned 1.19':
lidar invert = 2413.67
interpolated invert = 2412.48
END DESCRIPTION:
XS GIS Cut Line= 4
2278606.08200797508045.4899712032277914.55548338508099.808545413
2277582.34877714507966.0987061572277078.65510767508093.332181654
#Sta/Elev= 30
       0 2433.56      26 2433.49   198.7 2432.58   246.7 2428.69   269.3  2420.1
   318.9 2413.31     359 2411.38   369.8 2412.99   387.1 2417.86   455.3 2420.31
   563.2 2415.87   579.7 2412.48   631.8 2412.88   655.9  2418.3   730.7 2418.09
   773.8 2413.34   847.1 2413.56   854.3 2416.19  1006.7 2419.67  1043.5 2419.82
  1051.1  2420.2  1206.7 2419.88  1224.1 2424.41  1235.5 2424.98  1260.3 2418.94
  1305.7 2431.42  1398.6 2430.31  1421.2 2435.56  1433.6  2440.6  1571.3 2517.49
#Mann= 13 ,-1,0
       0     .05       0      26      .1       0   318.9     .04       0
   369.8     .08       0   563.2    .035       0   854.3      .1       0
  1006.7     .08       0  1043.5    .016       0  1051.1     .07       0
  1224.1    .016       0  1235.5     .07       0  1421.2    .016       0
  1433.6     .01       0
#XS Ineff= 2 , 0
                         1233.13         2438.02
Permanent Ineff=
       F       F
Bank Sta=563.2,854.3
XS Rating Curve= 0 ,0
Exp/Cntr=0.3,0.1

Type RM Length L Ch R = 1 ,260568  ,450.8,439.8,420.9
BEGIN DESCRIPTION:
channel burned 1.43':
lidar invert = 2410.53
effective invert = 2409.10
END DESCRIPTION:
XS GIS Cut Line= 4
2278787.03058561507257.9449111852278108.68449801507569.240718506
2277927.48246091507569.2407185062276933.19435991507903.767556225
#Sta/Elev= 30
       0 2473.73    55.9 2459.37   104.1 2435.95   161.5 2418.96   390.4 2418.12
   403.6 2413.53   434.4 2418.08   538.5 2417.65   592.9 2411.34   663.3 2418.01
  740.93 2412.83   750.9 2409.16   882.9  2409.1   902.9 2412.76  1028.1 2417.02
    1045 2413.19  1171.6 2414.78  1291.1 2416.76  1302.4 2416.64  1386.9  2418.7
  1395.3 2419.14  1526.1 2418.01  1568.3  2423.6    1588 2417.73  1602.1  2417.3
  1728.7 2416.01  1740.7 2420.22    1754 2420.81  1821.5 2450.91  1976.6 2535.25
#Mann= 13 ,-1,0
       0      .1       0   663.3     .12       0  740.93    .035       0
   902.9     .08       0  1171.6     .07       0  1291.1    .016       0
  1302.4     .07       0  1386.9    .016       0  1395.3     .07       0
    1588    .016       0  1602.1      .1       0  1740.7    .016       0
    1754      .1       0
#XS Ineff= 2 , 0
          650.82 2435.58 1566.96         2436.43
Permanent Ineff=
       F       F
Bank Sta=740.93,902.9
XS Rating Curve= 0 ,0
Exp/Cntr(USF)=0,0
Exp/Cntr=0.3,0.1

Type RM Length L Ch R = 1 ,260129  ,199.5,203.2,225.6
BEGIN DESCRIPTION:
channel burned 1.24':
lidar invert = 2407.75
interpolated invert = 2406.51
END DESCRIPTION:
XS GIS Cut Line= 2
2278410.02293876506993.1877736022276793.80817753507504.193833394
#Sta/Elev= 30
       0 2468.23    27.1 2458.77   183.1 2444.44   207.5 2435.79   232.7 2444.79
   266.2  2444.7   331.7 2439.16   352.1 2433.89   375.3 2410.58   387.9 2406.51
   522.1 2406.61  546.35 2410.51   580.9 2413.81   601.8 2414.53   681.6 2408.89
   723.5 2414.18   853.6 2415.91   884.4 2413.61   995.1 2415.71  1046.5 2419.56
  1252.1  2415.7    1285 2420.77  1298.2  2420.5  1319.2 2414.49  1440.9 2415.08
  1491.2 2424.32  1636.6  2438.4  1650.6 2439.91  1667.4 2442.12  1695.1 2451.26
#Mann= 11 ,-1,0
       0      .1       0   375.3    .035       0  546.35      .1       0
   580.9    .016       0   601.8      .1       0   884.4     .08       0
   995.1      .1       0    1285    .016       0  1298.2      .1       0
  1636.6    .016       0  1650.6      .1       0
#XS Ineff= 2 , 0
                         1290.93         2434.46
Permanent Ineff=
       F       F
Bank Sta=375.3,546.35
XS Rating Curve= 0 ,0
Exp/Cntr(USF)=0,0
Exp/Cntr=0.3,0.1

Type RM Length L Ch R = 1 ,259925  ,326.4,339.8,382.1
BEGIN DESCRIPTION:
channel burned 1.86':
lidar invert = 2407.16
effective invert = 2405.30
END DESCRIPTION:
XS GIS Cut Line= 3
2278437.02535534506799.0897935342277101.16646738507152.514408255
2276690.79203188507273.616046069
#Sta/Elev= 30
       0 2510.38      34 2498.27    71.2 2478.58   112.6 2466.51   253.3 2446.33
   427.1 2435.55   451.9 2428.88   472.32410.892   472.6 2410.57   480.8  2405.3
   625.7 2405.47   644.1 2410.57   675.3 2413.57   727.6 2413.44   764.8 2419.65
   787.7  2412.5   836.8 2412.52   861.5 2407.97   894.6 2411.95   919.4 2410.35
   964.4 2414.33    1147 2416.44    1358 2414.64  1376.6 2419.15  1389.6 2418.76
  1399.5 2414.92  1428.7 2414.48  1599.7 2424.95    1729 2438.78  1809.7 2452.03
#Mann= 8 ,-1,0
       0      .1       0   253.3     .12       0   472.3      .1       0
   472.6    .035       0   644.1     .08       0   861.5      .1       0
  1376.6    .016       0  1389.6      .1       0
#XS Ineff= 2 , 0
                         1387.28          2431.9
Permanent Ineff=
       F       F
Bank Sta=472.6,644.1
XS Rating Curve= 0 ,0
Exp/Cntr=0.3,0.1

Type RM Length L Ch R = 1 ,259586  ,280.5,272.8,242.4
BEGIN DESCRIPTION:
channel burned 0.85':
lidar invert = 2406.09
interpolated invert = 2405.24
END DESCRIPTION:
Node Name=U
XS GIS Cut Line= 3
     2278274.585      506551.2832277428.12173594506662.398248491
2276702.73528978506925.260739473
#Sta/Elev= 30
       0 2489.25    22.6 2486.46      68 2468.27      93 2462.11   288.9 2440.79
     305  2434.8   341.3 2411.15   357.5 2410.28  364.732407.377   369.6 2405.24
     543 2405.24   547.1 2407.38   563.7 2412.27   581.1 2412.61   672.1 2410.54
     773 2412.55   785.1 2412.01   797.2 2408.09   809.3 2408.12   841.6 2412.87
   887.7 2412.63   940.2  2409.2  1074.5 2413.68  1262.1 2413.41    1276 2417.07
  1291.9 2417.47  1304.6 2413.77  1338.7 2413.58  1381.2 2424.32  1625.3 2438.15
#Mann= 6 ,-1,0
       0      .1       0  364.73    .035       0   547.1     .08       0
   581.1      .1       0    1276    .016       0  1291.9      .1       0
#XS Ineff= 2 , 0
                         1280.79         2434.83
Permanent Ineff=
       F       F
Bank Sta=364.73,547.1
XS Rating Curve= 0 ,0
Exp/Cntr=0.3,0.1

Type RM Length L Ch R = 1 ,259313  ,228.8,221.3,246.3
BEGIN DESCRIPTION:
channel from lidar:
lidar invert = 2404.94
effective invert =2405.20
END DESCRIPTION:
XS GIS Cut Line= 4
2278173.63910122506250.3632174732277805.67198938506338.714418724
2277529.85593997506403.0459829722276651.99581905506725.876702145
#Sta/Elev= 30
       0 2564.94    46.8 2548.88   104.3 2523.44   141.4 2509.96   170.2 2502.11
   203.1 2487.97   275.6 2443.16   297.7 2423.14   308.7 2407.05   314.1 2404.94
   453.9  2406.6   503.2 2406.49   523.7 2409.76   540.1 2407.93   554.9 2409.74
   622.3  2405.7   635.8 2410.36   692.7 2412.41   730.1 2411.67   751.9 2407.92
   804.1 2409.02     851 2412.35  1153.6 2411.81    1213  2414.8  1221.7 2416.88
    1238 2417.06  1247.3 2415.38  1300.3 2415.22  1362.4 2425.24    1597 2437.45
#Mann= 6 ,-1,0
       0      .1       0   308.7    .035       0   453.9      .1       0
   804.1     .08       0  1221.7    .016       0    1238      .1       0
#XS Ineff= 2 , 0
                         1227.72         2439.35
Permanent Ineff=
       F       F
Bank Sta=308.7,453.9
XS Rating Curve= 0 ,0
Exp/Cntr(USF)=0,0
Minor Loss Coefficient=0
Exp/Cntr=0.3,0.1

Type RM Length L Ch R = 1 ,259092  ,480.1,509.9,510.1
XS GIS Cut Line= 4
2278029.69899466506026.700300136 2277658.0025083 506156.79407036
2276981.83420775506172.4248660382276371.49643402506188.583839939
#Sta/Elev= 30
       0  2616.7    86.4 2555.22   138.1  2514.1   154.2 2503.77   213.5 2456.12
   226.2 2442.81   249.7 2423.45   260.1 2406.85   263.7 2405.16   277.1 2402.98
   354.7 2402.97   384.42405.139   403.5 2408.83     439 2407.06   479.7 2408.86
   491.7 2405.53   531.7 2403.55   563.7 2409.78   583.5 2410.59   604.2 2406.72
   799.7 2407.56   831.7 2412.63  1031.8 2409.86  1060.8 2417.27  1331.9 2420.94
  1462.3 2427.63    1524  2427.1    1548  2430.8    1608 2432.85  1680.7 2439.25
#Mann= 9 ,-1,0
       0      .1       0   263.7    .035       0   384.4    .035       0
  384.42    .025       0     457     .08       0   747.8      .1       0
  1043.9     .06       0  1246.5     .05       0    1335      .1       0
#Block Obstruct= 2 ,-1
 1153.14 1199.89 2439.37  1444.2 1467.05 2447.73
Bank Sta=263.7,384.4
XS Rating Curve= 0 ,0
Exp/Cntr(USF)=0,0
Exp/Cntr=0.3,0.1

Type RM Length L Ch R = 1 ,258582  ,519.7,537.4,557.8
XS GIS Cut Line= 2
     2278036.505      505630.8422276466.75297633505688.328410656
#Sta/Elev= 30
       0 2636.32    24.3  2626.9    44.4  2616.7    76.4 2595.94   120.4 2570.66
   212.5 2513.71   280.6 2467.02   336.6 2419.88   355.2 2408.14   371.9 2403.07
   396.4 2401.25   540.7 2401.22   552.32403.164   564.7 2405.35   625.3 2405.61
   650.2  2410.2   840.9  2407.5   872.9 2408.26   896.9 2411.61   944.7 2412.19
   956.3 2415.82     985 2417.78    1049 2417.59  1109.1 2420.68  1237.2 2419.92
  1369.5 2422.36    1439 2425.71  1469.3 2430.77  1521.3 2434.36  1570.8  2440.9
#Mann= 6 ,-1,0
       0      .1       0     240     .12       0     340      .1       0
   371.9    .035       0   552.3     .08       0     730      .1       0
Bank Sta=371.9,552.3
XS Rating Curve= 0 ,0
Exp/Cntr=0.3,0.1

Type RM Length L Ch R = 1 ,258044  ,702.6,860.8,901.3
XS GIS Cut Line= 3
2278052.93002505505167.1521754412277016.82606934505037.058405217
2276909.96332952504972.011520105
#Sta/Elev= 30
       0 2513.08    56.2 2494.55    80.1 2484.47   113.6 2466.76   125.7 2458.52
   174.1 2430.82   190.2 2422.21   206.4 2415.63   226.5 2410.84   250.7 2407.57
   327.3 2405.82   346.3 2401.29   362.8 2399.91   557.1 2399.82  562.49 2401.25
   569.2 2403.98   577.3 2405.06   617.6 2404.81   650.7 2406.76   782.9 2406.14
   800.8 2405.42   819.1 2402.47   855.4 2405.11   883.6  2415.6   940.1 2415.72
   984.4 2419.48  1050.4 2427.83  1097.9 2437.77  1134.9 2448.24  1169.3 2460.23
#Mann= 7 ,-1,0
       0      .1       0     260    .025       0   346.3    .035       0
  562.49     .08       0     750     .05       0     850      .1       0
 1054.24     .05       0
Bank Sta=346.3,562.49
XS Rating Curve= 0 ,0
Exp/Cntr(USF)=0,0
Exp/Cntr=0.3,0.1

Type RM Length L Ch R = 1 ,257184  ,540.2,594.9,610.4
XS GIS Cut Line= 2
2278234.13206215504781.5170708482277402.46117393504019.539273822
#Sta/Elev= 30
       0  2453.2    51.5  2440.7   149.1 2422.59   181.7 2413.38     214 2397.68
   252.2 2404.77   355.8 2405.22   392.3 2397.66   448.9 2401.55   533.9 2397.41
   577.7  2396.2   588.6  2398.1   616.3 2404.22   634.1 2405.08   702.5 2401.16
   709.4 2397.77     717 2395.93     817 2395.66   825.5 2397.26   842.5 2407.25
     865 2411.58   886.9 2438.74   927.4 2478.25   941.2  2496.6   958.5 2526.99
   995.4 2565.85  1036.7 2594.51  1093.1 2641.98  1111.4 2652.09    1128 2655.97
#Mann= 6 ,-1,0
       0      .1       0   533.9    .035       0   588.6      .1       0
   709.4    .035       0   825.5    .025       0   941.2      .1       0
Bank Sta=533.9,825.5
XS Rating Curve= 0 ,0
Exp/Cntr(USF)=0,0
Exp/Cntr=0.3,0.1

Type RM Length L Ch R = 1 ,256589  ,522.2,445.5,406.6
XS GIS Cut Line= 2
     2278437.112      504321.6512277993.08564262503701.991405272
#Sta/Elev= 30
       0 2433.07    30.1 2429.79    56.5 2419.12   109.9 2404.17   138.4  2401.8
   144.3 2395.01   147.2 2394.04   246.6 2396.88   261.4 2394.51   276.2 2395.09
   276.2 2395.08     286 2393.12   320.4 2393.09   327.9 2394.86   338.1 2398.05
     350  2399.1   365.1 2394.79   373.7 2393.05   502.5 2392.81   514.2 2395.36
   522.8 2397.48   537.1 2404.72   556.6 2406.15   561.6 2408.06   597.3 2444.02
     626  2468.9   640.3 2487.48   700.5 2542.71   749.2 2586.63   762.3 2595.95
#Mann= 6 ,-1,0
       0      .1       0   276.2    .035       0   327.9      .1       0
   365.1    .035       0   514.2    .025       0   700.5      .1       0
Bank Sta=276.2,514.2
XS Rating Curve= 0 ,0
Exp/Cntr=0.3,0.1

Type RM Length L Ch R = 1 ,256143  ,625.5,543.7,481.9
XS GIS Cut Line= 3
2279023.98709566503895.2532611972278768.44576129503808.136897208
2278164.43897096503457.348338211
#Sta/Elev= 30
       0  2612.9    33.6 2591.07   126.6 2535.43   151.9 2519.35   164.6 2512.89
   206.3 2488.43   261.8 2459.46   284.2 2448.86   330.4 2424.25   367.4 2407.94
   385.9 2403.63   411.3 2400.85   424.5 2394.12   432.2 2391.04   442.1 2389.98
     641 2389.85   649.8 2390.16   658.2 2394.49   670.3 2402.78   687.9 2404.24
   705.1 2412.72   734.7 2434.85   761.7 2452.55   788.4 2473.42   807.8 2485.98
     830 2498.57   853.1 2508.82   862.4 2510.74   922.5 2531.63   968.5 2544.52
#Mann= 5 ,-1,0
       0      .1       0   424.5    .035       0   658.2      .1       0
  709.98    .025       0  819.98      .1       0
Bank Sta=424.5,658.2
XS Rating Curve= 0 ,0
Exp/Cntr(USF)=0,0
Exp/Cntr=0.3,0.1

Type RM Length L Ch R = 1 ,255599  ,555.3,512,469.6
XS GIS Cut Line= 3
     2279128.276      503101.3462278432.76280706503213.316696632
2278177.81117869503326.436581268
#Sta/Elev= 30
       0 2655.63    40.6 2625.76    81.1  2591.1    97.3 2579.81   125.6 2562.91
     150    2545     179 2520.73     231 2482.32   304.5  2431.7   326.1 2418.05
   336.4 2411.86   364.7 2399.61   376.9 2391.15   380.9 2388.96     389 2387.97
   506.5 2388.04   518.7 2390.83   526.8 2394.84   534.9 2396.78   559.2 2397.92
   591.6 2401.83   652.4 2400.03   668.6 2403.21   692.9 2403.63   710.9 2415.69
   744.5 2431.55     783 2452.94   804.8 2463.41   845.1 2479.74   983.4 2529.22
#Mann= 3 ,0,0
       0      .1       0   376.9    .035       0   518.7      .1       0
Bank Sta=376.9,518.7
XS Rating Curve= 0 ,0
Exp/Cntr=0.3,0.1

Type RM Length L Ch R = 1 ,255087  ,523,500.4,475.5
XS GIS Cut Line= 2
     2278848.877      502425.354     2278132.191      502986.123
#Sta/Elev= 30
       0 2702.68    45.2 2665.22    68.8 2648.48   122.8 2603.21   163.4 2576.05
     188 2563.81   214.1 2544.97   259.7 2504.88   272.3 2491.34   300.5 2473.61
   325.9 2460.81   361.5 2427.09   382.7 2399.48     397 2390.25   408.7 2387.09
     506 2387.14   516.1 2390.01   529.1 2395.99   561.7 2397.66   579.9 2396.71
   600.2 2399.74   635.8 2401.06   746.9 2394.84   761.2 2401.65     778 2403.08
   792.5 2421.13   801.1 2428.02   854.2 2452.65   864.3 2455.52     910 2475.55
#Mann= 4 ,-1,0
       0      .1       0     397    .035       0   516.1    .025       0
     560      .1       0
Bank Sta=397,516.1
XS Rating Curve= 0 ,0
Exp/Cntr=0.3,0.1

Type RM Length L Ch R = 1 ,254587  ,513.6,500,483.1
XS GIS Cut Line= 2
      2278379.22      502007.667     2277851.054      502748.707
#Sta/Elev= 30
       0 2689.95     5.2 2686.54    17.6 2674.03    54.9 2644.71    90.3 2623.09
   126.6 2598.29   138.1 2588.29     150 2582.12   188.5 2554.01   212.6 2533.56
   258.5 2509.82   276.9 2497.75   301.5 2473.98   316.2 2446.76   338.8 2431.38
   360.4  2407.2   375.2  2395.2   391.2 2387.43   399.7 2385.78   517.6 2385.78
     531 2387.32   559.6 2394.79   657.2 2392.12   685.8 2394.03   701.3 2400.34
   720.3  2401.4   740.3 2414.74   757.5 2422.98   832.3 2452.07     910 2484.81
#Mann= 7 ,-1,0
       0     .12       0      90      .1       0     150     .12       0
     210      .1       0     340     .05       0   391.2    .035       0
     531      .1       0
Bank Sta=391.2,531
XS Rating Curve= 0 ,0
Exp/Cntr=0.3,0.1

Type RM Length L Ch R = 1 ,254087  ,510.3,499.1,483.9
XS GIS Cut Line= 2
      2277878.81      501723.381     2277482.374      502542.489
#Sta/Elev= 30
       0 2677.88     6.3  2675.5    24.4  2657.7    99.8 2599.75   123.1 2573.73
   150.1 2555.29   157.5 2548.57   170.9 2543.85     180  2534.4     202 2517.51
   250.9 2483.83   264.2 2479.42   330.8  2439.8   341.7 2430.61   357.5 2412.25
   388.6 2388.92   397.5 2385.56   406.4 2383.94   530.4  2383.9   544.1 2385.57
   557.3 2386.85   570.8 2384.97   606.4 2391.09   629.2 2388.57   644.2 2391.03
   659.7 2398.77   681.9 2400.84     701 2413.58   786.5 2454.24     910 2522.07
#Mann= 3 ,-1,0
       0      .1       0   397.5    .035       0   544.1      .1       0
Bank Sta=397.5,544.1
XS Rating Curve= 0 ,0
Exp/Cntr=0.3,0.1

Type RM Length L Ch R = 1 ,253588  ,513.8,500.9,491.1
XS GIS Cut Line= 2
     2277352.553      501529.522     2277071.455       502395.02
#Sta/Elev= 30
       0  2664.1    29.1 2641.67    45.9  2635.5    75.3 2612.22   104.8 2585.87
   125.8 2570.93     151 2545.73   176.3  2527.4   188.9 2510.19   226.7 2486.87
     254 2462.01   314.3 2420.26   327.7 2417.33   365.1 2395.32   373.9 2388.02
   382.4 2384.88   390.8 2382.34   490.9 2382.22   546.4 2382.23   555.6 2384.56
     580  2389.7   630.5 2388.14   647.3 2390.61   660.3 2397.27     681 2397.65
   689.4 2408.07   697.8 2414.01   815.5  2472.7   861.8 2489.99     910 2503.46
#Mann= 4 ,-1,0
       0      .1       0   382.4    .035       0   555.6    .025       0
     580      .1       0
Bank Sta=382.4,555.6
XS Rating Curve= 0 ,0
Exp/Cntr=0.3,0.1

Type RM Length L Ch R = 1 ,253087  ,501.7,500,501.7
XS GIS Cut Line= 2
     2276808.687      501392.325     2276644.674      502287.422
#Sta/Elev= 30
       0 2670.41    28.7  2648.5    41.5 2636.61    57.8 2629.24    70.1 2618.14
   122.9 2579.65   147.3 2559.63   159.5 2547.28     173 2540.96   208.3 2506.79
   220.5 2501.64   240.8 2482.79   289.6  2443.7   301.8 2435.82   313.9 2424.28
   330.3 2416.94   373.8 2381.36   379.2 2379.84   505.1    2381   562.1 2380.99
   590.5 2379.05   610.9 2381.54     619 2385.45   631.2 2387.63   646.4 2394.44
   671.9 2396.13   692.2 2402.79   749.1 2426.62   856.9 2484.65     910  2508.2
#Mann= 4 ,-1,0
       0      .1       0     300    .025       0   373.8    .035       0
   505.1      .1       0
Bank Sta=373.8,505.1
XS Rating Curve= 0 ,0
Exp/Cntr=0.3,0.1

Type RM Length L Ch R = 1 ,252587  ,507.7,499.3,488.9
XS GIS Cut Line= 2
     2276308.262      501306.046     2276159.669      502203.832
#Sta/Elev= 30
       0 2695.08    34.1 2666.73    76.2  2634.9    84.3 2625.19    96.7 2620.53
   124.8 2595.96   161.3 2567.51   177.5 2550.18   197.8 2542.08     214  2525.7
   266.7 2480.27   282.9 2463.47   300.1  2453.7   354.1 2394.63   361.1 2388.45
     373 2381.76   385.5 2378.13   513.8 2378.06   546.5 2378.67   558.6 2381.58
   570.8 2385.89   587.2 2388.38   627.6 2390.01   643.8 2388.59   668.1 2393.48
   692.4 2394.35   704.6 2402.16   716.8 2405.25   838.4 2470.63     910 2503.08
#Mann= 4 ,-1,0
       0      .1       0     290    .025       0     373    .035       0
   558.6      .1       0
Bank Sta=373,558.6
XS Rating Curve= 0 ,0
Exp/Cntr=0.3,0.1

Type RM Length L Ch R = 1 ,252088  ,316.9,319.2,322.7
XS GIS Cut Line= 2
      2275776.59      501234.533     2275702.126      502141.482
#Sta/Elev= 30
       0 2598.11    14.7 2593.52    50.8  2577.1    62.9 2567.34      77 2562.21
    86.9 2553.35   123.1 2527.26   139.1 2511.97   151.2 2507.04   159.8 2498.81
   223.4 2451.23   235.4 2440.61   247.5 2436.75   267.5 2423.33   307.7 2403.84
   323.7 2400.56   339.8 2393.16   355.8 2390.13   371.9 2380.13   379.9 2377.22
     445 2377.19   551.8 2377.27   562.1 2380.16   588.6 2385.57   640.8 2386.84
     701 2393.04     713 2401.37   738.3 2409.12   757.2 2417.63     910 2500.61
#Mann= 4 ,-1,0
       0      .1       0     360    .025       0   371.9    .035       0
   562.1      .1       0
Bank Sta=371.9,562.1
XS Rating Curve= 0 ,0
Exp/Cntr=0.3,0.1

Type RM Length L Ch R = 1 ,251768  ,383.1,395.7,409.7
XS GIS Cut Line= 3
2275582.95074559501258.1669019032275440.91473566501492.526318285
2275375.57817109502070.612878694
#Sta/Elev= 30
       0 2521.06     5.4 2519.19    22.2 2505.31    74.8 2469.85    87.7 2464.97
    97.4 2457.17   141.1 2429.11   164.4 2417.48   202.2 2401.83   218.7 2400.42
     243 2394.28   265.4  2393.6   335.1 2384.52   367.3 2383.03   382.9 2378.54
   396.5 2376.49   423.7 2376.34   548.4 2376.36   555.3 2378.26   560.5 2381.33
   576.6 2382.51   592.7 2385.62     633 2384.82   649.1    2389   673.2 2390.37
   677.2  2391.7   681.3 2393.72   689.3 2401.09   788.9 2464.93   855.8 2505.04
#Mann= 6 ,-1,0
       0      .1       0     160     .06       0  274.04      .1       0
  374.04    .025       0   382.9    .035       0   555.3      .1       0
Bank Sta=382.9,555.3
XS Rating Curve= 0 ,0
Exp/Cntr(USF)=0,0
Exp/Cntr=0.3,0.1

Type RM Length L Ch R = 1 ,251373  ,286.6,287.9,292.8
XS GIS Cut Line= 3
 2275279.3013601501118.7963940432275077.30255024501415.826872924
2274927.66314074502049.875515731
#Sta/Elev= 30
       0 2485.28    41.4 2455.03    75.4 2433.25    85.1 2427.42   138.3 2400.84
   150.8 2399.94   172.2 2395.14   204.7 2391.72   286.1  2389.6   367.9 2389.87
   404.5 2383.46   463.3 2382.92   479.8 2377.28     488 2374.72   656.5 2375.07
   664.7 2375.26   670.5 2377.41   680.5  2381.6   697.6 2384.78   738.7 2384.83
   753.6 2387.45   771.6 2387.98   789.9 2398.83   808.6 2411.62     862 2454.16
   902.8 2482.42   927.8 2493.94   960.6 2504.37   976.4 2506.61  1010.7 2517.62
#Mann= 5 ,-1,0
       0      .1       0     220     .06       0     330      .1       0
   479.8    .035       0   670.5      .1       0
#XS Ineff= 2 , 0
          360.79 2402.75
Permanent Ineff=
       F       F
Bank Sta=479.8,670.5
XS Rating Curve= 0 ,0
Exp/Cntr=0.3,0.1

Type RM Length L Ch R = 1 ,251085  ,426.4,458.3,481.3
XS GIS Cut Line= 3
2274990.74446394500958.7410080762274835.91688087501211.102214969
     2274637.851      501991.459
#Sta/Elev= 30
       0 2458.08    54.5 2421.65    68.6 2417.59    82.6 2409.74   115.5 2395.99
   128.7 2396.09   148.3 2391.26   186.9  2388.6   284.4 2387.77   298.2 2389.77
   413.8 2390.32   429.2 2389.11   450.9 2382.07   521.4  2381.7   537.1 2377.07
   554.1 2374.16   698.5 2374.29   706.8 2376.79   735.7 2385.44   764.5 2384.41
   776.9 2381.99     788 2385.28   809.9 2387.39   916.4 2478.79   933.7 2510.62
     942    2518     963 2530.05   995.6 2544.65  1057.9  2568.7  1101.2 2582.81
#Mann= 7 ,-1,0
       0      .1       0      80     .06       0     270     .08       0
     280      .1       0  486.07    .025       0   537.1    .035       0
   706.8      .1       0
#XS Ineff= 2 , 0
          406.99 2418.47
Permanent Ineff=
       F       F
Bank Sta=537.1,706.8
XS Rating Curve= 0 ,0
Exp/Cntr=0.3,0.1

Type RM Length L Ch R = 1 ,250627  ,488,541,583.3
XS GIS Cut Line= 3
2274715.56193326500764.7494241162274264.70561715501478.857494835
2274233.32181324501828.988759955
#Sta/Elev= 30
       0 2436.61     5.7 2435.73    66.7 2402.88    81.1  2401.8    90.4 2396.88
   118.8 2391.72     171 2387.47   330.4  2389.1   355.3 2383.01   383.7 2383.21
     400 2388.72   466.7 2388.59   492.8 2379.15   582.7  2381.4   643.6 2379.52
     661 2375.03   687.1 2372.41     781 2374.84   795.2 2383.59   818.9  2385.8
   833.1 2402.67   862.9 2431.62   909.8 2463.33   925.9 2490.61   940.1 2507.89
   987.4  2539.1  1015.5 2566.29  1095.8 2598.46  1156.7  2629.6  1196.1  2645.4
#Mann= 6 ,-1,0
       0      .1       0     120     .06       0     300     .08       0
     400      .1       0     661    .035       0     781      .1       0
#XS Ineff= 2 , 0
          428.62 2420.85
Permanent Ineff=
       F       F
Bank Sta=661,781
XS Rating Curve= 0 ,0
Exp/Cntr=0.3,0.1

Type RM Length L Ch R = 1 ,250086  ,483.5,498.8,510.5
XS GIS Cut Line= 2
2274575.10199192500701.399592036     2273592.669      501144.322
#Sta/Elev= 30
       0  2404.1    30.3 2395.21    48.1 2390.03   130.5 2385.02   191.9 2384.32
   219.8  2386.2   244.5 2384.46   349.9 2386.59   393.7 2383.83   450.8 2383.75
   503.4 2376.84   540.4 2376.56   556.1 2373.62   569.2 2371.25   603.9 2371.19
   676.5 2371.28   683.3 2373.76   700.9 2381.61   715.8 2383.47   733.9  2403.6
   744.7  2413.4   781.3 2440.34   879.1 2512.81   888.2 2523.45   903.3 2545.22
   963.8 2583.77   999.2 2610.16  1047.5 2640.29  1060.5 2655.84  1077.7 2667.22
#Mann= 7 ,-1,0
       0      .1       0    30.3     .06       0   130.5      .1       0
   556.1    .035       0   683.3      .1       0   733.9    .025       0
   781.3      .1       0
#XS Ineff= 2 , 0
          350.47 2393.02
Permanent Ineff=
       F       F
Bank Sta=556.1,683.3
XS Rating Curve= 0 ,0
Exp/Cntr=0.3,0.1

Type RM Length L Ch R = 1 ,249587  ,485.1,501.6,516.9
XS GIS Cut Line= 2
2274377.82193595500343.240472013     2273401.001      500606.838
#Sta/Elev= 30
       0 2420.54    26.6 2406.31    34.9 2400.32    51.4 2398.44    63.9 2392.37
    92.9 2383.99   101.1 2382.63   159.1 2382.83   205.2 2380.76   237.7 2382.59
   304.2 2381.21   399.4 2381.75   428.4 2375.75     445 2374.91   456.4 2371.02
   461.6 2370.06     590 2370.09   596.7 2370.96   623.2 2373.28   639.7 2379.22
   656.3 2380.78   660.5  2382.7   681.6 2397.52   691.9 2406.81   710.2 2425.97
   747.5 2445.43   782.6  2466.3   867.8 2513.34   952.4 2564.18  1011.8  2604.3
#Mann= 8 ,-1,0
       0      .1       0      20     .06       0     130      .1       0
     430    .025       0   456.4    .035       0   596.7      .1       0
     630    .025       0     740      .1       0
#XS Ineff= 2 , 0
          395.38 2396.11
Permanent Ineff=
       F       F
Bank Sta=456.4,596.7
XS Rating Curve= 0 ,0
Exp/Cntr=0.3,0.1

Type RM Length L Ch R = 1 ,249085  ,467.8,487.8,506.2
XS GIS Cut Line= 2
2274295.72387729499947.719765339     2273293.743      500036.123
#Sta/Elev= 30
       0 2443.42    71.8 2410.02     120 2398.99   136.1  2393.4   163.3 2391.84
   184.3 2384.11   204.3  2379.5   224.4 2377.79     337 2378.91   405.1 2377.06
     440 2378.97   473.4 2375.09   485.4 2370.79   497.5 2368.25   617.9 2368.25
     626 2370.66     630 2372.73     642 2378.51   662.1 2381.62   710.3 2421.93
   722.3  2436.4   730.4 2439.32   753.7 2441.36   778.6 2446.88   862.9 2490.65
   930.8 2542.23   947.2 2549.28   963.3 2559.44   991.4 2584.81  1005.9 2604.05
#Mann= 8 ,-1,0
       0      .1       0      40     .06       0     140      .1       0
     340     .08       0     440      .1       0   485.4    .035       0
     626    .025       0     630      .1       0
#XS Ineff= 2 , 0
          354.25 2393.34
Permanent Ineff=
       F       F
Bank Sta=485.4,626
XS Rating Curve= 0 ,0
Exp/Cntr=0.3,0.1

Type RM Length L Ch R = 1 ,248597  ,484.9,511.8,533.9
XS GIS Cut Line= 2
2274296.41093595499583.343351991     2273295.527       499449.37
#Sta/Elev= 30
       0 2426.08    20.4 2418.57    52.7 2410.17   105.2 2403.07     202 2393.66
   222.2 2390.32   238.3 2389.76   286.8 2377.41   319.1 2375.72   403.8 2376.41
     424 2373.65   448.2 2374.09   468.3 2368.26   482.6 2368.01   504.7 2366.69
   601.6 2366.67   607.2 2367.91   629.8 2375.55   641.9 2376.02   645.9 2378.05
     654 2386.31   666.1 2395.09   682.3 2413.62   687.3 2417.53   819.5 2503.11
   847.7  2524.9   856.4 2529.68   927.5 2582.32   984.5 2626.57  1009.8 2647.84
#Mann= 6 ,-1,0
       0      .1       0     140     .06       0     240      .1       0
   482.6    .035       0   607.2    .025       0     740      .1       0
Bank Sta=482.6,607.2
XS Rating Curve= 0 ,0
Exp/Cntr=0.3,0.1

Type RM Length L Ch R = 1 ,248086  ,451.5,497.1,538.6
XS GIS Cut Line= 2
2274377.70346663499235.109586652     2273471.529      498836.288
#Sta/Elev= 30
       0  2428.1    67.2 2404.83    93.4  2399.6   237.7 2386.93   324.3 2374.18
   378.9 2374.09     402 2370.66   442.7 2372.86   457.8 2368.34   482.1 2364.62
   591.3 2364.66   600.4 2368.17   622.2 2376.34   639.9  2378.3   661.1  2395.3
   700.9 2420.17   770.4 2480.65   783.9 2500.92     822 2535.42   842.2 2561.13
   871.4 2592.77   876.6 2601.69   888.8  2639.3   901.9 2651.59   915.1 2654.83
   931.2 2651.69   946.4  2646.7   958.5  2638.5   976.2 2636.72   990.1 2628.81
#Mann= 7 ,-1,0
       0      .1       0     240     .06       0     350      .1       0
   457.8    .035       0   600.4    .025       0     670      .1       0
     890     .06       0
Bank Sta=457.8,600.4
XS Rating Curve= 0 ,0
Exp/Cntr=0.3,0.1

Type RM Length L Ch R = 1 ,247588  ,497,501.5,506.5
XS GIS Cut Line= 2
2274531.72223197499090.778759955     2273924.252      498272.774
#Sta/Elev= 30
       0 2436.86    80.9 2414.69   109.5 2409.73   158.1 2405.66   195.2 2396.64
   269.6  2387.3     321 2372.01   418.2 2373.35   455.4 2367.81   489.7 2370.47
   506.9  2365.3   529.8    2362   609.8    2362   621.2 2365.35   644.1 2374.07
   659.7 2374.88   669.9 2381.52   675.6 2389.97   689.6 2429.33   694.5 2435.97
   714.5 2456.27   744.4 2482.06   792.8 2527.96     849 2583.06   875.7 2604.18
   904.3    2632   915.7 2639.12   923.7 2640.86     950 2635.55  1018.9 2607.32
#Mann= 8 ,-1,0
       0      .1       0     200     .06       0     330      .1       0
   506.9    .035       0   621.2      .1       0     700    .025       0
     790      .1       0     950     .06       0
Bank Sta=506.9,621.2
XS Rating Curve= 0 ,0
Exp/Cntr=0.3,0.1

Type RM Length L Ch R = 1 ,247087  ,493.8,500,507.9
XS GIS Cut Line= 2
     2274857.618      498735.396     2274360.091      497973.447
#Sta/Elev= 30
       0 2421.74   100.9 2404.25     150 2392.42   184.7 2386.95   199.2 2379.33
   216.5 2377.95   246.3 2369.62   317.9 2373.02   340.8 2369.65   370.5 2369.24
   394.4 2363.33   403.9 2362.82   421.7 2360.54   513.8 2360.56   522.9 2363.02
     544 2369.69   574.9 2372.87   580.7 2376.65   592.2 2393.69   604.6 2416.09
   618.2 2430.84   661.9 2467.01   713.6 2512.29   747.9 2537.83   794.5 2579.93
   814.8 2595.09   824.3 2609.13   862.5 2646.93   898.6 2679.57     910 2688.07
#Mann= 6 ,-1,0
       0      .1       0     120     .06       0     360      .1       0
   403.9    .035       0   522.9    .025       0     590      .1       0
Bank Sta=403.9,522.9
XS Rating Curve= 0 ,0
Exp/Cntr=0.3,0.1

Type RM Length L Ch R = 1 ,246587  ,499.5,500,501.5
XS GIS Cut Line= 2
     2275259.969      498512.051     2274830.811      497709.602
#Sta/Elev= 30
       0 2428.99      42 2420.62    89.4 2406.33   134.8 2397.52   175.6 2386.55
     200 2377.22   216.5    2376   225.5 2372.75   257.3  2368.5     289 2366.85
   316.2 2369.53   341.9 2369.73   375.2 2365.58   388.8  2362.7   402.4 2359.84
   522.1 2359.87   534.1 2362.61   548.7 2370.35   561.2 2372.19   570.3 2381.41
   579.3 2392.43   597.5  2408.6   607.8 2415.11   642.8 2442.27   683.7 2463.58
   705.4 2471.27   751.7 2483.77   792.5 2492.98   856.2 2504.47     910  2518.6
#Mann= 7 ,-1,0
       0      .1       0      90     .06       0     200      .1       0
   388.8    .035       0   534.1    .025       0     540     .12       0
     650      .1       0
Bank Sta=388.8,534.1
XS Rating Curve= 0 ,0
Exp/Cntr=0.3,0.1

Type RM Length L Ch R = 1 ,246087  ,520,500.4,484
XS GIS Cut Line= 2
     2275699.626      498280.637      2275276.05      497475.229
#Sta/Elev= 30
       0  2441.3    34.7 2433.63    80.7 2419.43   107.9 2413.26   139.5 2401.31
   162.1 2400.22   171.1 2395.04   198.2 2386.83   206.5    2383   220.8 2380.63
   229.9 2376.99   238.9 2376.65     248 2373.15   262.8 2372.62   275.1 2368.59
   295.5 2366.01   325.4 2368.83   392.6 2364.37     399 2361.69   410.7 2359.13
   470.1 2359.12   550.8 2359.16   561.9 2361.69   586.9  2370.7   612.3 2372.95
   618.6 2377.41   627.6 2387.13   643.3 2394.97   654.7 2398.44     910 2424.76
#Mann= 7 ,-1,0
       0      .1       0     160     .06       0     270      .1       0
     380    .025       0     399    .035       0   561.9    .025       0
     720      .1       0
Bank Sta=399,561.9
XS Rating Curve= 0 ,0
Exp/Cntr=0.3,0.1

Type RM Length L Ch R = 1 ,245587  ,490.6,479.7,471.2
XS GIS Cut Line= 2
     2276207.372       497991.91     2275641.677      497278.949
#Sta/Elev= 30
       0 2517.21    39.2 2505.25    50.2 2500.23    69.5 2495.38   109.6 2473.61
     121 2463.99     138 2454.68   161.8 2439.14   177.9 2434.25   223.9 2411.02
   263.9 2396.88   274.1 2391.58   289.4 2390.86   308.9 2381.25   330.3  2373.7
   359.1 2369.46   371.1 2360.09   381.3 2357.45   462.6 2357.41   488.6 2357.41
   526.4 2359.98   590.8 2366.94   672.4 2368.79   730.2 2367.33   787.2 2361.14
   807.1  2368.4   835.6  2369.8     847    2374   856.2 2381.61   910.1 2393.65
#Mann= 5 ,-1,0
       0      .1       0     190     .07       0     290     .08       0
   371.1    .035       0   526.4      .1       0
Bank Sta=371.1,526.4
XS Rating Curve= 0 ,0
Exp/Cntr=0.3,0.1

Type RM Length L Ch R = 1 ,245107  ,487.5,486,484.1
XS GIS Cut Line= 4
     2276591.502      497636.9622276171.71822153497200.723134314
2275873.42184371496900.5728887012275715.44699384496904.436998904
#Sta/Elev= 30
       0  2542.2    38.6 2536.47    78.6 2542.97    91.3 2540.27   105.2 2532.34
   118.2 2516.18   146.5 2501.08   157.8 2492.38   169.1 2488.56     237 2442.57
   249.5 2438.68   270.2 2424.97   333.2 2392.28   347.3 2390.29   375.6 2373.05
   393.8 2369.32   408.6 2360.37   420.2 2356.31   532.6 2356.31     551 2360.17
     577 2364.74   644.4 2364.26   695.6 2368.96   780.7 2364.87   826.1 2358.81
  1033.8 2375.35  1053.8 2381.69  1077.8 2384.03  1097.8 2391.08  1186.6 2400.44
#Mann= 5 ,-1,0
       0      .1       0     240     .06       0     390      .1       0
   408.6    .035       0     551      .1       0
Bank Sta=408.6,551
XS Rating Curve= 0 ,0
Exp/Cntr=0.3,0.1

Type RM Length L Ch R = 1 ,244621  ,727.6,574.2,399.4
XS GIS Cut Line= 3
2276927.42994403497275.2305866522276524.30724274 496871.47518138
2275863.70053875496813.915709366
#Sta/Elev= 30
       0 2469.75   132.9 2427.33   144.2 2426.59   168.8 2417.13   279.9 2386.36
   308.1 2369.86   334.7 2367.55   353.3 2359.09   361.3 2355.57   387.3 2355.31
   464.8 2355.32   497.1 2358.99   525.4 2357.74   610.8 2364.38     643 2362.25
   739.3 2364.57   791.5 2362.59   823.6 2356.03   855.8 2356.67   891.9 2363.41
     912 2357.85     928 2356.51   956.1 2361.38  1036.4 2362.45  1088.6 2367.88
  1108.7 2367.13  1120.8  2370.1    1177 2370.99  1217.1 2374.72  1233.7 2378.93
#Mann= 4 ,-1,0
       0      .1       0     170     .06       0   353.3    .035       0
   497.1      .1       0
Bank Sta=353.3,497.1
XS Rating Curve= 0 ,0
Exp/Cntr=0.3,0.1

Type RM Length L Ch R = 1 ,244047  ,271.4,277.6,287
XS GIS Cut Line= 3
2276781.58576803496231.3681759962276458.60041873496680.721229277
2275877.26412541      496773.609
#Sta/Elev= 30
       0 2479.12      94 2461.43   140.2 2429.93   154.9 2416.46   171.4 2408.33
   185.7 2405.06   204.2 2396.47   223.9 2394.71   235.4 2385.94   248.8 2384.55
  284.22 2356.76   292.9 2354.09   425.9 2354.25   437.9 2356.52   450.5    2357
   468.4 2357.92   480.9 2354.91   516.4 2361.89   543.8 2362.15     755 2363.11
   778.6  2361.4   793.4 2354.33   823.2 2353.98   855.6 2355.68   867.8    2361
   894.7 2359.37     965 2363.24   989.3 2367.81  1090.3 2370.27  1142.1 2375.58
#Mann= 8 ,-1,0
       0      .1       0   185.7     .06       0  284.22    .035       0
   437.9      .1       0   450.5    .025       0   543.8      .1       0
   793.4     .06       0   894.7      .1       0
Bank Sta=284.22,437.9
XS Rating Curve= 0 ,0
Exp/Cntr=0.3,0.1

Type RM Length L Ch R = 1 ,243769  ,210.2,235.7,281.8
BEGIN DESCRIPTION:
xs 4
END DESCRIPTION:
XS GIS Cut Line= 3
2276597.99157459496051.6614280772276199.92145316496548.673834019
2275769.63756468  496661.4220187
#Sta/Elev= 30
       0 2469.46    50.7 2455.97    96.3 2440.49   124.5 2425.93     156 2402.57
   167.4 2396.87   194.9 2393.76   252.8 2382.16     267 2374.18   290.8 2375.27
   319.7 2360.96     342 2355.15   350.4 2353.19     526 2354.67     540 2353.57
     581 2362.45   643.5 2363.26   657.2 2362.78   673.7 2353.62   694.4 2352.67
   712.3 2356.94   777.1 2360.39   789.5 2365.36   814.3 2367.22   938.4 2367.81
   967.3 2370.48     988    2375  1033.5 2394.66  1046.5 2398.05  1081.6 2398.92
#Mann= 7 ,-1,0
       0      .1       0     280     .08       0     290     .07       0
     342    .035       0     526    .025       0     540      .1       0
  916.77     .06       0
Bank Sta=342,526
XS Rating Curve= 0 ,0
Exp/Cntr(USF)=0,0
Exp/Cntr=0.5,0.3

Type RM Length L Ch R = 1 ,243533  ,110.7,105.5,94.8
BEGIN DESCRIPTION:
structure xs 3
END DESCRIPTION:
XS GIS Cut Line= 4
2276578.16856488496023.7777706462276219.01773913496191.761253672
2275963.88027653496404.5994298852275730.82682175496632.797750981
#Sta/Elev= 30
       0 2469.33    38.7 2460.33    71.8 2450.84    86.8 2445.11   119.9 2427.38
     171 2385.98   182.7 2379.79   205.3 2374.19     223 2367.87   245.1 2363.73
   360.6 2360.48     405 2359.69   419.4  2354.7   429.9 2352.34     586 2352.47
   654.7 2351.35   671.1 2354.39   686.7 2357.81   704.7 2361.42   740.3 2366.03
   779.9 2366.36   840.3 2366.99   867.6 2368.72   879.5 2370.71   901.5 2371.03
   912.5 2375.83   969.1 2394.13   981.1 2396.36  1051.4 2397.74  1054.9 2397.81
#Mann= 9 ,-1,0
       0      .1       0     171     .07       0   360.6      .1       0
   419.4    .035       0   671.1     .07       0   686.7    .025       0
   779.9     .07       0   969.1     .06       0  1051.4      .1       0
#XS Ineff= 2 , 0
             379 2362.43     711         2366.32
Permanent Ineff=
       F       F
Bank Sta=419.4,671.1
XS Rating Curve= 0 ,0
Exp/Cntr=0.5,0.3

Type RM Length L Ch R = 1 ,243428  ,346,340.9,340.6
BEGIN DESCRIPTION:
structure xs 2
END DESCRIPTION:
XS GIS Cut Line= 3
2276549.46098291 495954.601030862276162.09928565496095.316096395
2275690.94097633496530.109838217
#Sta/Elev= 30
       0 2476.22    49.8 2460.35   103.5 2446.92   124.8    2439   143.5 2428.12
   159.8 2414.71   171.6 2407.72   201.4 2382.78   221.5 2370.67   239.7 2362.57
   262.1 2360.86   363.1 2361.38     442 2359.17     468 2354.04   473.9  2353.1
   686.2 2351.13   706.4 2352.83   721.6 2357.03   733.4 2363.88   822.4 2366.08
   850.2 2369.79   863.1 2376.89   886.7  2380.5   904.6 2379.62   915.5 2384.36
   939.8 2386.58   958.3  2391.8   972.5  2393.7   992.3 2395.31  1053.2 2399.29
#Mann= 10 ,-1,0
       0      .1       0   363.1     .07       0     468    .025       0
   473.9    .035       0   706.4     .07       0   733.4      .1       0
   822.4     .07       0   863.1     .06       0   972.5     .07       0
   992.3     .06       0
#XS Ineff= 2 , 0
             458 2361.85     722          2364.8
Permanent Ineff=
       F       F
Bank Sta=473.9,706.4
XS Rating Curve= 0 ,0
Exp/Cntr(USF)=0,0
Exp/Cntr=0.5,0.3

Type RM Length L Ch R = 1 ,243087  ,534.1,485.3,424.9
XS GIS Cut Line= 2
     2276124.104      495669.881     2275453.355      496284.858
#Sta/Elev= 30
       0 2491.33    40.4 2463.65    70.2 2438.47   105.5 2412.53   118.4 2404.71
   164.7 2367.22   186.3 2353.28     217 2352.62   229.8 2356.79   257.1 2357.65
   316.5 2354.63   363.5 2355.16   387.3 2352.39   401.4 2349.97     509 2349.91
     548 2349.95   557.2 2352.59   571.3 2360.73     577 2362.07   614.5 2359.75
   645.7 2361.05   721.1 2359.91   738.4 2363.39   772.3 2363.79   786.2 2369.14
   797.8 2371.34   835.6 2386.64   857.3 2393.18     879 2396.81     910 2398.36
#Mann= 8 ,-1,0
       0      .1       0     310    .025       0   387.3    .035       0
   557.2     .05       0     610      .1       0     660     .05       0
     750      .1       0     800     .05       0
Bank Sta=387.3,557.2
XS Rating Curve= 0 ,0
Exp/Cntr=0.3,0.1

Type RM Length L Ch R = 1 ,242602  ,560.5,511.8,459.9
XS GIS Cut Line= 2
     2275517.794      495257.5352275261.99459109496225.931884668
#Sta/Elev= 30
       0 2657.66    24.5    2644   112.3 2584.62   169.3 2534.85   210.9 2507.02
   231.3 2489.15   260.3 2470.94   285.1  2461.1   297.5    2453   330.6 2418.67
   347.2 2394.76   355.4  2379.1   359.6  2368.2   367.8 2357.71   376.1 2351.38
   388.5  2349.2     397 2347.22   524.7 2347.26   531.2 2349.39     554 2356.62
   578.8 2351.79   609.8 2351.96   636.8 2353.17     674 2358.64   818.8 2357.54
   847.8 2358.89   876.7  2363.3   905.7 2362.55     973 2391.15  1001.6 2397.52
#Mann= 7 ,-1,0
       0      .1       0     340    .025       0   388.5    .035       0
   531.2    .025       0     550     .08       0     750     .05       0
     850      .1       0
Bank Sta=388.5,531.2
XS Rating Curve= 0 ,0
Exp/Cntr=0.3,0.1

Type RM Length L Ch R = 1 ,242090  ,523,502.9,484.1
XS GIS Cut Line= 2
     2274772.253      495293.3872275041.66574967496226.308521627
#Sta/Elev= 30
       0 2557.91    25.6 2537.17    37.3 2530.76    61.1 2512.59    95.5 2491.59
   135.5 2470.98   145.1 2466.22   187.1 2451.38     208 2440.54   262.1 2424.86
   282.9 2416.86     312 2402.55   341.2 2381.33   353.7 2368.65     362 2356.56
     368 2351.34   374.5 2347.96   378.7 2346.25   511.9 2346.28   526.7 2347.93
   553.5 2353.49   628.5 2351.62   695.1 2355.24   803.3 2356.13     820 2357.71
     845 2361.18   869.9 2360.32   924.1 2378.41   949.5 2389.89     971 2397.64
#Mann= 5 ,-1,0
       0      .1       0   374.5    .035       0   526.7      .1       0
     610     .05       0     820      .1       0
Bank Sta=374.5,526.7
XS Rating Curve= 0 ,0
Exp/Cntr=0.3,0.1

Type RM Length L Ch R = 1 ,241587  ,499.8,500,502.1
XS GIS Cut Line= 2
     2274232.431      495536.293     2274652.172      496343.707
#Sta/Elev= 30
       0 2586.09    95.7 2540.27   131.7 2528.46   175.5 2509.72   196.2 2491.71
   217.4 2476.02   230.9 2461.36   240.7  2446.4   250.9  2437.1   271.5 2415.16
   298.5 2392.35   325.6 2371.54   343.6 2360.78   357.1 2350.03   366.2 2347.32
   387.6 2344.91   531.4 2344.98   545.8 2347.17   555.5 2349.35   578.1  2348.8
   600.6  2352.2   699.8 2355.79   726.8  2358.8   749.4 2358.75   753.9 2359.75
   763.2 2367.25   783.5 2379.07   821.5 2397.37   875.5 2411.95     910 2418.72
#Mann= 5 ,-1,0
       0      .1       0   366.2    .035       0   545.8      .1       0
     710     .06       0     720      .1       0
Bank Sta=366.2,545.8
XS Rating Curve= 0 ,0
Exp/Cntr=0.3,0.1

Type RM Length L Ch R = 1 ,241087  ,525.9,500.9,477.3
XS GIS Cut Line= 2
     2273790.962      495763.523     2274204.514      496574.124
#Sta/Elev= 30
       0 2577.05    55.7 2545.65    78.2 2530.91   109.2  2513.3   135.9 2494.64
   216.2 2442.86   269.7 2413.13   280.3 2405.01   289.3 2396.43   302.7 2380.71
   316.2 2368.13   323.3 2359.65   340.2 2348.04   356.6 2343.03   558.2 2342.94
   567.7 2343.08   578.6 2347.75   585.6 2351.55   599.1 2353.53   639.5 2354.57
   666.5 2353.91   684.4 2356.34   711.4 2355.39   720.3 2356.45   733.6 2365.01
   751.5 2373.97   778.7  2389.9   796.7 2402.38     830 2423.06     910 2470.83
#Mann= 3 ,0,0
       0      .1       0   340.2    .035       0   578.6      .1       0
Bank Sta=340.2,578.6
XS Rating Curve= 0 ,0
Exp/Cntr=0.3,0.1

Type RM Length L Ch R = 1 ,240586  ,516.7,497.3,479.2
XS GIS Cut Line= 2
     2273284.855      496065.897     2273849.428      496779.592
#Sta/Elev= 30
       0  2576.3    64.5 2527.35    76.3 2520.63   101.5 2501.01   127.9 2484.31
   157.2 2462.48   177.6 2451.52   246.7 2410.33   308.4 2376.71   321.3 2370.63
   334.2 2361.58     351    2346   356.1  2343.4   366.3 2341.25   531.5 2341.24
   540.1  2341.6   544.8 2343.26   548.6 2345.96   554.3 2348.55   579.9 2351.41
   641.7 2352.07     657 2350.44   682.5 2353.88   705.2 2354.81   710.9 2357.39
   743.7 2378.14   815.1 2425.33   870.4 2455.63   891.6 2465.66     910 2472.62
#Mann= 3 ,0,0
       0      .1       0     351    .035       0   548.6      .1       0
Bank Sta=351,548.6
XS Rating Curve= 0 ,0
Exp/Cntr=0.3,0.1

Type RM Length L Ch R = 1 ,240089  ,531.9,501.5,468.7
XS GIS Cut Line= 2
     2272849.416      496427.445     2273516.311      497047.198
#Sta/Elev= 30
       0 2597.45    47.5 2559.15    73.9 2540.23    85.7 2534.04    96.6 2523.86
   113.6 2515.69   125.9 2503.08   145.7 2488.38   200.3 2452.92   214.1 2442.81
   263.6  2413.7   320.2 2377.64   331.4 2367.35   342.3 2349.55   345.6  2345.6
   351.3  2342.3   365.5 2339.74   472.6 2339.66   543.8 2340.98   552.3 2345.64
   555.3 2347.29   664.5 2352.03   693.8 2348.33   702.3  2348.8   716.4 2352.03
   735.5 2352.47   795.8 2381.52   828.3 2394.53   846.6 2398.69   910.4 2407.13
#Mann= 3 ,0,0
       0      .1       0   345.6    .035       0   552.3      .1       0
Bank Sta=345.6,552.3
XS Rating Curve= 0 ,0
Exp/Cntr=0.3,0.1

Type RM Length L Ch R = 1 ,239587  ,521.1,500.3,475.7
XS GIS Cut Line= 2
     2272487.555      496932.522     2273293.808      497354.559
#Sta/Elev= 30
       0 2631.37    39.5 2606.18    59.4 2591.44    68.4 2581.84      82 2556.35
    86.5 2552.14   131.6 2519.67   163.2 2494.78   187.7 2479.26   242.9 2439.49
   285.4 2414.13   352.9 2369.89   370.9 2356.03   379.9 2344.95   384.5 2341.83
     398 2337.94   533.5 2337.88   551.5 2337.88   562.1 2341.03   570.7 2341.99
   610.2 2348.34     647 2346.18   682.8 2350.13   732.1 2348.21   745.7 2350.11
   768.2 2349.92   795.3 2354.78   842.6 2378.67   866.3 2387.62     910 2395.96
#Mann= 4 ,-1,0
       0      .1       0   384.5    .035       0   562.1    .025       0
   570.7      .1       0
Bank Sta=384.5,562.1
XS Rating Curve= 0 ,0
Exp/Cntr=0.3,0.1

Type RM Length L Ch R = 1 ,239087  ,509.3,498.6,486.2
XS GIS Cut Line= 2
     2272259.987      497476.499     2273133.574      497731.342
#Sta/Elev= 30
       0 2621.33    41.9 2625.27    66.9  2624.1    79.4 2617.78   104.4 2598.87
   123.3 2582.97   133.5 2567.89   145.9 2555.41   159.5 2527.93   162.7 2522.46
   168.4 2515.94   187.8 2498.99   204.4  2481.9   216.9 2467.17   241.9 2445.91
   250.2 2434.31     362  2339.8   375.2 2336.25   541.9 2336.28   554.4 2340.27
   636.2 2349.99   683.5 2349.27     721 2345.63   741.9 2345.82   758.5 2349.66
   800.7  2348.5   808.5 2350.55   829.4 2363.51   839.4 2367.39     910 2378.06
#Mann= 3 ,0,0
       0      .1       0     362    .035       0   554.4      .1       0
Bank Sta=362,554.4
XS Rating Curve= 0 ,0
Exp/Cntr=0.3,0.1
