HEC-RAS study GRNBRRRV.prj: GRNBRRRV

--- GRNBRRRV.g01 (geometry) --- (continued)

Type RM Length L Ch R = 1 ,213270  ,65.9,57.5,58.1
BEGIN DESCRIPTION:
structure xs 3
END DESCRIPTION:
XS GIS Cut Line= 4
2264629.14814217486711.3356274562264308.64507217486576.386966404
2263862.70595462486642.8352534342263331.15202029486189.617574749
#Sta/Elev= 30
       0  2490.8      36  2468.4    70.5 2442.34   139.8 2397.88   230.2 2330.98
   261.5 2308.89   274.2 2296.97   283.2  2291.9   330.9 2289.67   344.5 2285.27
   353.1  2280.4   360.4 2276.57   368.5 2275.28   542.2  2275.4     553 2280.11
   562.6 2284.24   586.8 2287.67   647.5 2288.63   744.6 2288.51     781 2292.46
     830 2292.36   854.5 2291.96     980 2293.94  1110.9  2296.4  1285.5 2303.71
  1368.4 2308.12    1430 2314.64  1460.8 2314.83  1473.2 2320.08  1497.2 2325.18
#Mann= 12 ,-1,0
       0      .1       0   230.2     .06       0   344.5     .08       0
   353.1    .035       0     553     .06       0   647.5     .05       0
   744.6     .06       0     830     .05       0   854.5     .06       0
     980     .05       0  1110.9      .1       0  1285.5     .06       0
#XS Ineff= 3 ,-1
       0     331 2290.48     575  797.75 2288.79  797.75  1497.2 2309.05
Permanent Ineff=
       F       F       F
Bank Sta=353.1,553
XS Rating Curve= 0 ,0
Exp/Cntr(USF)=0,0
Exp/Cntr=0.5,0.3

Type RM Length L Ch R = 1 ,213213  ,211.4,209.6,207.7
BEGIN DESCRIPTION:
structure xs 2
END DESCRIPTION:
XS GIS Cut Line= 4
2264650.83631984486636.6319043742264332.74304736486516.142028434
2263850.34558123486584.1234798192263375.09362299486148.593492698
#Sta/Elev= 30
       0 2474.18    41.3 2449.23   100.9 2416.89   228.1 2333.92   250.9 2317.36
   263.8 2308.53   276.6 2296.89   285.2 2292.64   360.9 2287.31     369 2285.88
   381.1 2279.07   393.2 2275.16   562.9 2275.19  576.91 2278.88   591.2 2284.76
   607.1 2286.86   660.2 2288.37   740.6 2286.85   793.1 2288.45   821.4 2292.35
   867.7 2292.66   997.4 2294.11  1057.4 2294.85  1128.2 2296.22  1210.6 2299.66
    1349  2310.8  1371.7 2311.85  1399.9 2319.72  1441.5 2331.88  1471.9 2335.47
#Mann= 13 ,-1,0
       0      .1       0   250.9     .06       0   360.9    .025       0
   381.1    .035       0  576.91     .06       0   660.2     .05       0
   867.7     .06       0   997.4     .05       0  1057.4     .06       0
  1128.2      .1       0  1210.6     .06       0    1349      .1       0
  1399.9     .06       0
#XS Ineff= 3 ,-1
     1.2   374.22290.145     585  824.79    2288  824.79  1471.9 2315.64
Permanent Ineff=
       F       F       F
Bank Sta=381.1,576.91
XS Rating Curve= 0 ,0
Exp/Cntr(USF)=0,0
Exp/Cntr=0.5,0.3

Type RM Length L Ch R = 1 ,213003  ,254,300.9,340.9
BEGIN DESCRIPTION:
xs 1
END DESCRIPTION:
XS GIS Cut Line= 4
2264696.94487922486424.5633684712264327.13217045486302.747283196
2263833.07144982486381.0221114312263387.61742705486072.292220328
#Sta/Elev= 30
       0 2430.59      85 2390.27   202.6 2326.68   236.7 2309.33   270.3 2294.81
   278.8 2294.38   288.4 2290.22   295.6 2289.19   408.6 2289.78   424.8 2287.14
   453.22278.333   461.2 2274.94   465.3 2274.81   656.3 2274.91   667.7 2277.96
   694.7 2285.98   716.3 2287.85   862.5 2286.47   890.7 2290.84   913.1 2291.92
   939.3 2293.05   968.5 2291.74   994.6 2293.98  1075.6 2294.55  1177.2 2300.79
  1198.3 2306.33  1254.5 2310.62  1301.2 2329.61  1338.5 2339.13  1431.6 2346.85
#Mann= 10 ,-1,0
       0      .1       0     180     .06       0     290    .025       0
   453.2    .035       0   667.7     .06       0  797.94     .05       0
  897.94     .06       0 1000.78     .05       0 1020.78     .06       0
 1270.78      .1       0
#XS Ineff= 2 , 0
                          901.41         2309.75
Permanent Ineff=
       F       F
Bank Sta=453.2,667.7
XS Rating Curve= 0 ,0
Exp/Cntr=0.3,0.1

Type RM Length L Ch R = 1 ,212702  ,401.6,478.5,533.3
XS GIS Cut Line= 4
2264777.03197917486263.8299667662264506.69917323486104.457611428
2263804.99739074485988.3963718192263547.59890917485903.402115639
#Sta/Elev= 30
       0 2424.41    28.8 2408.16    87.3 2381.45    98.5 2374.71   115.5 2372.26
   149.6 2355.34   177.4 2349.88   228.5 2328.22   288.9 2296.68   303.4 2294.98
   320.4 2287.05   340.7 2285.97   433.9 2289.56   524.1 2288.68   592.1 2282.78
   607.6 2277.44   616.4 2274.39     823 2274.44   839.4 2277.45     872 2284.58
   948.9 2291.58   985.3 2297.35  1055.4 2304.78  1063.8 2308.48  1080.7 2310.24
  1107.4 2320.49    1127 2324.99  1194.4 2330.21  1221.4 2343.76  1296.1  2359.5
#Mann= 8 ,-1,0
       0      .1       0     260     .06       0  403.81      .1       0
  603.81    .025       0   607.6    .035       0   839.4      .1       0
  903.81    .025       0 1003.81      .1       0
Bank Sta=607.6,839.4
XS Rating Curve= 0 ,0
Exp/Cntr=0.3,0.1

Type RM Length L Ch R = 1 ,212224  ,503.2,514.7,523.8
XS GIS Cut Line= 2
2264779.99906409486082.0669646892264040.11778282485370.827671021
#Sta/Elev= 30
       0 2368.95    76.9 2337.62    88.5 2331.13    99.6 2329.84   116.7 2322.39
   151.4 2312.68   161.8 2307.84   180.2 2306.99   249.4 2287.72   299.4 2285.68
   405.3 2288.59   480.3 2286.07   509.7 2286.37   569.1 2274.99   587.9 2274.82
   687.8 2273.66   722.8 2274.71   732.2 2278.36   748.8 2287.99     770 2289.33
   775.6 2290.91   787.6 2301.37     792 2308.98   803.9 2333.02   809.3 2338.37
   861.3 2364.56   872.8 2368.88   902.9 2386.21   959.5 2410.72  1026.3 2450.09
#Mann= 6 ,-1,0
       0      .1       0      70     .06       0     210     .05       0
     510      .1       0   587.9    .035       0   722.8      .1       0
Bank Sta=587.9,722.8
XS Rating Curve= 0 ,0
Exp/Cntr=0.3,0.1

Type RM Length L Ch R = 1 ,211709  ,543.7,535.5,528.1
XS GIS Cut Line= 2
2265086.73820248485773.9568139092264452.63126451484993.007090827
#Sta/Elev= 30
       0 2373.34    26.8 2359.08    39.3 2349.76    56.4  2346.4    83.4 2331.52
   105.6 2311.91   118.3 2306.34   179.6 2307.54   200.8  2306.2   213.5 2304.03
   243.2  2293.3     296  2287.7     334 2284.64   434.6 2284.24   485.8 2276.19
     499 2277.84   508.4 2275.85   526.6 2272.47     664 2272.44   673.5 2275.54
   693.4 2284.65   713.3 2288.89   737.8 2320.35     773 2347.89   789.3  2367.2
     810 2383.57   861.5 2407.96   898.8 2428.53   949.1 2453.02    1006 2484.44
#Mann= 8 ,-1,0
       0      .1       0      50     .06       0     280     .05       0
     300      .1       0   508.4    .035       0   673.5      .1       0
     680    .025       0     750      .1       0
Bank Sta=508.4,673.5
XS Rating Curve= 0 ,0
Exp/Cntr=0.3,0.1

Type RM Length L Ch R = 1 ,211174  ,575.5,579,582.7
XS GIS Cut Line= 2
2265461.05522729485330.9645081952264839.63822729484666.178508195
#Sta/Elev= 30
       0 2341.61    40.8 2319.43    64.1 2308.41    89.6 2298.66   109.4 2293.83
   155.8 2288.38   276.6 2286.81   336.4 2282.88   369.3 2282.75   399.6 2273.98
   412.2 2271.44   592.9 2271.44   604.6 2273.89   616.3 2277.03   632.1 2284.94
   645.6 2285.91   651.5 2287.82   666.9 2304.75   681.1 2318.88   727.6  2356.5
   737.7 2362.57   760.3 2379.17   774.5 2387.15   780.3 2391.52   796.4 2400.43
   807.3 2404.52   821.4 2412.82   862.1 2441.28   879.9 2455.45     910 2476.06
#Mann= 6 ,-1,0
       0     .05       0     250      .1       0   399.6    .035       0
   604.6    .025       0     660     .05       0     790      .1       0
Bank Sta=399.6,604.6
XS Rating Curve= 0 ,0
Exp/Cntr=0.3,0.1

Type RM Length L Ch R = 1 ,210595  ,507.4,503.6,500.3
XS GIS Cut Line= 2
 2265966.0252809485050.088661052     2265246.355      484234.491
#Sta/Elev= 30
       0 2370.13    43.9 2339.45    89.8  2310.3   115.3 2295.79   129.2 2290.38
   139.9 2288.22   152.2 2287.67   251.9 2287.75     410 2284.72   462.3 2282.48
   483.7 2278.06   513.3 2280.06     524 2278.53   531.9 2274.62   537.6 2271.39
   545.3 2270.53     732 2270.53   737.4 2271.35   744.4 2274.76   758.7 2283.38
   764.1 2284.72   775.6 2285.09   780.1 2286.94   790.7 2295.18   801.1 2305.66
   806.7 2309.29   840.8 2325.79   965.5 2399.53  1057.5 2450.28  1087.7 2469.98
#Mann= 6 ,-1,0
       0      .1       0     130     .05       0     410      .1       0
   531.9    .035       0   744.4     .05       0     790      .1       0
Bank Sta=531.9,744.4
XS Rating Curve= 0 ,0
Exp/Cntr=0.3,0.1

Type RM Length L Ch R = 1 ,210091  ,490.7,495.8,501
XS GIS Cut Line= 2
2266347.99648338484696.9804709772265716.33588835484018.027090827
#Sta/Elev= 30
       0 2369.49      38 2346.45    81.8 2322.91   129.9 2299.46   147.2 2292.87
   158.2 2290.29   190.9 2286.65   240.1 2285.16   254.5 2286.06   265.8 2284.79
   311.1 2283.81   387.6 2283.81   475.2 2281.31   492.2 2281.76   500.7 2280.14
   506.4 2275.72     512 2271.01   518.8 2269.81   716.2 2269.84     722 2270.71
   729.9 2275.99   744.1 2284.51   764.6  2285.5   783.7 2301.92   797.4 2311.75
   851.2 2346.14     863 2352.62   906.7 2381.93   915.8 2389.07   927.3 2396.15
#Mann= 6 ,-1,0
       0      .1       0     190     .05       0     380      .1       0
   506.4    .035       0   729.9     .05       0     860      .1       0
Bank Sta=506.4,729.9
XS Rating Curve= 0 ,0
Exp/Cntr=0.3,0.1

Type RM Length L Ch R = 1 ,209595  ,560.8,534.3,512.2
XS GIS Cut Line= 2
2266691.35390075484374.705078421     2265999.804       483568.23
#Sta/Elev= 30
       0 2402.26    44.2 2375.52   119.6 2321.82   144.3 2307.38   165.4 2298.78
     197 2294.59   318.2 2283.68   447.3 2277.84   460.4 2273.12   497.3  2278.7
   502.6 2277.75   508.8 2273.34   514.9 2269.58   528.1 2269.13   713.4 2269.16
   718.2 2269.71   723.9 2272.72   723.9 2272.73   739.7 2276.45   757.9 2283.23
     773 2284.62   780.6 2288.13   808.2 2315.47   857.2 2353.16   877.5 2371.31
   908.3 2392.27   939.5 2409.81   993.4 2448.16  1044.4 2494.17  1062.4 2506.71
#Mann= 5 ,-1,0
       0      .1       0   508.8    .035       0   723.9      .1       0
     780     .05       0     800      .1       0
Bank Sta=508.8,723.9
XS Rating Curve= 0 ,0
Exp/Cntr=0.3,0.1

Type RM Length L Ch R = 1 ,209061  ,538,446.3,369.6
XS GIS Cut Line= 3
2267007.61941737483781.1978843612266551.63412406483456.996529023
2266115.85074391483459.364280902
#Sta/Elev= 30
       0 2437.46    43.5 2413.06   126.9 2362.43   244.7 2298.92   269.2 2286.66
     284  2283.8   298.7 2272.04   308.5 2268.79   318.3 2268.34     428 2268.49
   462.5 2271.59   490.1 2272.34   510.2 2270.18   534.3 2270.16   553.9 2274.76
     619 2271.89     643 2273.26     683 2270.14     695 2271.37     715  2283.1
     735  2286.3     743 2293.52   751.8 2307.43     771 2324.04     835 2367.49
     843 2371.09     871 2390.88     931 2429.53     963 2446.66   995.3 2460.14
#Mann= 6 ,-1,0
       0      .1       0     280    .025       0   298.7    .035       0
   462.5      .1       0  629.49    .025       0  729.49      .1       0
Bank Sta=298.7,462.5
XS Rating Curve= 0 ,0
Exp/Cntr=0.3,0.1

Type RM Length L Ch R = 1 ,208615  ,426.3,414.8,407.3
XS GIS Cut Line= 2
     2267163.724      483014.2442266177.36669429483245.018533007
#Sta/Elev= 30
       0 2483.47    69.4 2442.27    98.1 2422.33   159.7 2375.19   204.9 2352.58
   262.5 2314.26   274.8 2308.61   315.9 2299.54   344.6 2289.34   356.9 2277.77
   364.9 2272.03   373.4 2268.15   381.6 2267.59   484.3 2267.71   518.1 2271.49
   525.4 2273.96   566.4 2279.41   582.9 2276.84   619.8 2278.88   652.7 2275.59
   669.1 2276.26   681.5 2273.77   693.8 2268.81   734.9 2269.37   759.5  2283.5
   780.1 2283.86   800.6 2290.57   817.7 2302.72   837.6 2311.25    1013 2364.88
#Mann= 7 ,-1,0
       0      .1       0     300     .12       0     310      .1       0
   364.9    .035       0   518.1      .1       0     700    .025       0
     740      .1       0
Bank Sta=364.9,518.1
XS Rating Curve= 0 ,0
Exp/Cntr=0.3,0.1

Type RM Length L Ch R = 1 ,208200  ,383.5,333.9,300.7
XS GIS Cut Line= 2
2267005.18482233482593.7416610522266152.01782233482865.040508195
#Sta/Elev= 30
       0 2445.41    51.3 2408.54     107 2364.09   135.4 2342.57   156.3 2327.51
     169 2320.09   189.9 2305.84   210.5 2294.98   223.5 2286.69   236.1 2282.62
   261.3 2281.51   265.5 2279.66   273.9 2272.94   279.4 2269.85   286.5 2266.97
   290.2 2266.94   481.2 2267.04   496.3 2268.84   517.3 2268.25   529.9 2269.29
   546.7 2275.28   571.9 2278.75   601.3 2277.83   626.5 2282.93   639.1 2283.03
   726.5 2293.08   773.4 2302.44   816.5 2312.36   861.5  2324.9   895.3  2336.3
#Mann= 4 ,-1,0
       0      .1       0     240     .12       0   279.4    .035       0
   496.3      .1       0
Bank Sta=279.4,496.3
XS Rating Curve= 0 ,0
Exp/Cntr=0.3,0.1

Type RM Length L Ch R = 1 ,207866  ,348.8,348.8,349.6
XS GIS Cut Line= 2
2266831.70307434482139.9497343092266103.94422367482723.120733856
#Sta/Elev= 30
       0 2473.57    31.8 2446.91    80.2 2412.16    96.8 2403.02   111.5 2391.78
   122.9 2386.74   131.4 2380.44   189.1 2346.75   219.6 2326.37     231 2321.41
   262.3 2297.03   283.4  2283.2   296.5 2278.53     305 2271.79   312.1 2268.79
   327.4 2265.84   481.2 2265.94   494.5 2268.53   555.4 2276.52   588.9 2276.03
   612.3 2282.52   629.9 2283.84   665.8 2282.71   686.3 2284.93   731.9 2283.94
   782.4 2286.62   825.8 2296.31   882.7 2312.72   903.9 2320.43   932.6  2334.3
#Mann= 3 ,0,0
       0      .1       0   312.1    .035       0   494.5      .1       0
#XS Ineff= 2 , 0
                           650.6         2310.98
Permanent Ineff=
       F       F
Bank Sta=312.1,494.5
XS Rating Curve= 0 ,0
Exp/Cntr(USF)=0,0
Exp/Cntr=0.3,0.1

Type RM Length L Ch R = 1 ,207517  ,441.9,401.3,341.6
XS GIS Cut Line= 3
2266732.46716526481777.9061364662266125.63240134482258.029812729
2265873.12570669482587.276673458
#Sta/Elev= 30
       0 2550.49    16.8  2538.1    36.7 2519.57    51.4 2508.42    71.8  2498.3
    89.1 2493.83   119.3 2489.55   136.4 2482.41     218 2424.41     256 2404.98
   270.2 2395.07   291.1 2385.51   321.7  2363.6   379.2 2334.54   437.2 2309.29
   456.5 2290.62   483.8 2269.95   495.2 2264.94     637 2264.88   654.6 2269.92
   678.7 2280.29   733.7 2278.91   772.4 2282.57   788.5 2281.28     817 2283.49
   949.2 2282.69   999.6 2286.77    1026 2294.34  1107.4 2329.35  1188.7 2373.13
#Mann= 3 ,0,0
       0      .1       0   483.8    .035       0   654.6      .1       0
#XS Ineff= 2 , 0
                          749.74         2319.15
Permanent Ineff=
       F       F
Bank Sta=483.8,654.6
XS Rating Curve= 0 ,0
Exp/Cntr=0.3,0.1

Type RM Length L Ch R = 1 ,207116  ,319.7,308.6,290.3
XS GIS Cut Line= 2
2266138.16406203481577.6808387222265742.10583474482430.033599022
#Sta/Elev= 30
       0 2428.67    39.1 2404.23    56.8 2395.46    73.4 2385.12   172.8 2313.73
   184.7 2303.76   197.9 2284.93   202.3 2280.02   208.9 2274.43     220  2268.3
   228.8 2264.93   237.6 2263.88   378.8 2263.91   386.6 2264.89   396.4 2268.17
   436.1 2276.21   464.9 2278.37     507  2277.3   545.8 2277.64   573.3 2280.19
   603.7 2281.47     617 2280.66   633.5 2281.75   744.9 2281.53     772 2283.64
   793.4 2287.58   810.6 2293.02   841.9 2305.18   881.6 2322.65   939.9  2341.5
#Mann= 3 ,0,0
       0      .1       0     220    .035       0   396.4      .1       0
#XS Ineff= 2 , 0
                          542.17         2303.46
Permanent Ineff=
       F       F
Bank Sta=220,396.4
XS Rating Curve= 0 ,0
Exp/Cntr=0.3,0.1

Type RM Length L Ch R = 1 ,206807  ,237.6,216.5,190.1
XS GIS Cut Line= 2
2265805.31388664481483.5261076862265554.73633634482295.582983683
#Sta/Elev= 30
       0 2421.28     8.6 2412.59    14.3 2407.78    47.8 2383.63    56.1 2378.62
    82.2 2360.15   118.9 2339.08   135.7 2326.43   148.2 2315.97   160.8 2308.13
   169.2 2301.15   194.3 2272.98   206.8 2266.31   227.8 2263.03   357.5 2263.06
   374.3 2264.81   380.62266.333   395.2 2270.27     412  2270.7   428.7 2274.39
   459.7  2272.7   474.8 2275.66   554.3 2278.19     571 2280.81   596.2  2280.5
   633.8 2283.67   759.4 2299.86   788.7  2302.8   834.8  2310.9   849.8  2314.7
#Mann= 3 ,0,0
       0      .1       0   206.8    .035       0   380.6      .1       0
#XS Ineff= 2 , 0
                          538.73         2300.83
Permanent Ineff=
       F       F
Bank Sta=206.8,380.6
XS Rating Curve= 0 ,0
Exp/Cntr(USF)=0,0
Exp/Cntr=0.3,0.1

Type RM Length L Ch R = 1 ,206591  ,503.7,497.6,490.3
XS GIS Cut Line= 2
2265528.39621489481446.8362312782265465.53980993482272.383115639
#Sta/Elev= 30
       0 2418.26    14.4 2406.74    34.4 2389.14    42.5 2384.24    54.5 2373.68
    66.5 2364.28   110.7 2332.96   146.8 2310.14   182.9 2290.12   206.9 2271.51
   218.6 2266.18     227 2262.55     231 2262.44   367.4  2262.5   375.2 2263.03
   388.8 2266.31   423.6 2273.41   435.6 2274.61   455.7 2274.33   479.7 2276.38
   531.9 2276.85   551.9 2278.24     564 2280.27     588 2279.88   668.3 2285.91
   712.4 2287.32   728.4 2291.19   744.5 2296.89   792.6 2319.59   827.9 2333.54
#Mann= 4 ,-1,0
       0      .1       0     170    .025       0   218.6    .035       0
   388.8      .1       0
#XS Ineff= 2 , 0
                          540.45         2296.68
Permanent Ineff=
       F       F
Bank Sta=218.6,388.8
XS Rating Curve= 0 ,0
Exp/Cntr=0.3,0.1

Type RM Length L Ch R = 1 ,206093  ,503.8,500.9,497.2
XS GIS Cut Line= 2
2265012.75120248481424.853838722     2265003.579      482178.143
#Sta/Elev= 30
       0 2434.19    16.3 2421.25    48.3 2398.09    56.3 2391.24    68.3 2383.88
    96.3 2362.82   136.3 2331.11   148.3 2320.29     159 2308.98   164.3 2302.26
   188.3 2282.63   200.3 2270.35   204.3 2267.52   212.3 2265.44   216.3 2264.45
   220.3 2261.44   224.3 2261.09   404.4 2261.09   412.4 2262.04   420.9 2265.36
   428.4 2268.33   440.4 2271.22   464.4 2274.52   512.4 2275.29   548.4 2279.22
   564.4 2279.44   584.4 2285.95   592.4 2286.99   676.4  2312.6   753.3 2338.71
#Mann= 4 ,-1,0
       0      .1       0     190    .025       0   212.3    .035       0
   420.9      .1       0
Bank Sta=212.3,420.9
XS Rating Curve= 0 ,0
Exp/Cntr=0.3,0.1

Type RM Length L Ch R = 1 ,205592  ,489.3,496.3,506.4
XS GIS Cut Line= 2
      2264503.78481427.269838721     2264515.048      482180.563
#Sta/Elev= 30
       0  2426.1    13.7 2413.94    41.9 2392.34    89.9 2358.94    97.9 2350.05
   149.9 2318.86   169.9 2304.91   191.5  2286.6   209.9 2267.65   213.9 2265.34
   224.9 2262.89   229.9 2261.01   237.9 2260.22     390 2260.22     410 2262.45
     430 2269.34   448.3 2270.43     466 2273.93     478 2273.95     490 2272.31
     506  2272.6     510 2272.96     522 2277.92     526 2278.41     534 2278.38
     546 2274.53     562 2276.41   609.3 2294.48     694 2335.28   753.4 2362.29
#Mann= 4 ,-1,0
       0      .1       0     190    .025       0   224.9    .035       0
     410      .1       0
Bank Sta=224.9,410
XS Rating Curve= 0 ,0
Exp/Cntr=0.3,0.1

Type RM Length L Ch R = 1 ,205096  ,476.9,502.5,524.8
XS GIS Cut Line= 2
2264030.70840496 481415.89063624     2263984.285        482165.4
#Sta/Elev= 30
       0 2416.35    49.4 2375.57   101.7 2330.54   113.5  2323.6   125.5 2312.73
   165.3 2282.88   181.6 2268.18   189.7 2264.91   197.7 2260.29   201.7 2259.72
     394 2259.75   408.8 2264.55   426.1    2271   450.1 2274.22   470.2 2274.92
   479.1 2273.22   498.2 2272.97   510.3 2277.38   522.3 2278.08   538.3  2272.9
   546.3 2274.52   562.4 2274.97   578.4 2279.97   603.7 2293.78   642.5 2319.94
   646.5 2323.15   654.5 2335.24   658.5 2339.97   730.7 2391.27   750.9 2408.14
#Mann= 3 ,0,0
       0      .1       0   189.7    .035       0   408.8      .1       0
Bank Sta=189.7,408.8
XS Rating Curve= 0 ,0
Exp/Cntr=0.3,0.1

Type RM Length L Ch R = 1 ,204594  ,600.9,641.7,658.2
XS GIS Cut Line= 2
     2263620.976       481214.52     2263406.856       482098.97
#Sta/Elev= 30
       0 2431.98    31.5 2413.04    80.9 2391.45   138.5 2354.76   179.7 2331.23
   200.3 2317.76   216.7 2302.98   228.2 2295.34   245.6 2277.03   261.3 2269.89
   268.6  2263.7   274.4 2260.48   297.8 2259.08   306.6 2261.22   360.4 2261.08
   373.1 2259.25   550.1 2259.31  561.51 2264.04   587.1 2275.44   640.6 2273.36
   661.2 2276.88   677.7 2272.58   727.1 2276.54   747.7 2285.59   776.5 2303.19
   817.6 2332.49   834.5  2348.8     867 2370.62   883.5 2378.69     910 2386.11
#Mann= 5 ,-1,0
       0      .1       0   268.6    .035       0   306.6      .1       0
   360.4    .035       0  561.51      .1       0
Bank Sta=268.6,561.51
XS Rating Curve= 0 ,0
Exp/Cntr=0.3,0.1

Type RM Length L Ch R = 1 ,203952  ,390.2,402,417.9
XS GIS Cut Line= 2
2263112.23717637480995.5751586342262750.27790495481832.817398599
#Sta/Elev= 30
       0 2481.82    45.3 2449.23    88.9 2422.43   115.1 2401.64   156.4    2361
   193.5  2326.7   214.2 2305.36   253.8  2272.1     266 2267.92     272 2262.37
   276.3 2258.69   280.6 2257.85   459.3 2259.88     529 2258.17   533.4 2259.58
   536.7 2262.99   542.1 2269.99   546.5 2272.51   563.9 2275.71   597.6 2276.38
   664.5 2272.35   677.2 2275.92   688.9 2276.26   703.4 2271.64   768.7 2276.73
   799.2 2281.11   828.8 2296.19   899.5 2343.66   903.8 2348.39   912.1 2362.19
#Mann= 4 ,-1,0
       0      .1       0     240    .025       0     272    .035       0
   536.7      .1       0
Bank Sta=272,536.7
XS Rating Curve= 0 ,0
Exp/Cntr(USF)=0,0
Exp/Cntr=0.3,0.1

Type RM Length L Ch R = 1 ,203550  ,447.3,457.3,472.8
XS GIS Cut Line= 2
2262779.28448148480842.9800756942262313.01525198481693.097206235
#Sta/Elev= 30
       0 2465.81    29.9 2452.37   115.9 2396.75   153.1 2364.99   180.7  2343.4
     185 2339.04   198.7 2320.72   242.6  2282.7   253.4 2271.85   270.5 2262.29
   277.9 2258.35   285.4 2257.47     477 2257.59   484.1 2258.72   490.7 2262.38
   499.8 2268.96     518 2274.39   528.3 2275.67   559.1 2275.79   619.7 2272.22
   650.3 2275.44   666.8 2271.37   678.6 2272.68   746.8 2273.07   771.7 2276.66
   796.7  2288.7   855.4  2327.4   871.5 2339.69   879.8 2349.89   969.6 2418.99
#Mann= 4 ,-1,0
       0      .1       0     200    .025       0   270.5    .035       0
   490.7      .1       0
Bank Sta=270.5,490.7
XS Rating Curve= 0 ,0
Exp/Cntr(USF)=0,0
Exp/Cntr=0.3,0.1

Type RM Length L Ch R = 1 ,203093  ,471.6,499,527.4
XS GIS Cut Line= 2
2262393.38669429480659.4090660152261928.41344218 481339.37793797
#Sta/Elev= 30
       0 2372.86    51.8 2339.61    87.2 2314.13   142.7 2284.61   172.2 2274.96
     196  2261.5   203.6 2257.97   210.5 2257.03   399.3 2257.06   406.1 2257.71
   413.2 2261.25   420.2 2269.35   428.1 2271.23   491.6 2267.92   554.6 2270.25
   588.5 2270.03   598.2 2274.18   609.4 2274.92   627.3  2270.5   636.9 2272.76
   658.3 2274.58   698.6 2275.53   721.6  2277.7   738.7 2284.11   784.9 2310.75
   787.8  2314.3   796.4  2341.1   799.3 2345.22   813.7 2354.91   823.7 2358.44
#Mann= 5 ,-1,0
       0      .1       0     196    .035       0   413.2      .1       0
     430    .025       0     440      .1       0
Bank Sta=196,413.2
XS Rating Curve= 0 ,0
Exp/Cntr=0.3,0.1

Type RM Length L Ch R = 1 ,202594  ,416.5,499.1,568.1
XS GIS Cut Line= 2
     2262186.296      480262.123     2261521.644      480883.684
#Sta/Elev= 30
       0 2324.14    27.9  2318.9    52.2 2310.95   117.9 2283.14   139.8  2276.6
   227.2 2271.38   252.7 2273.97   323.5 2273.84   331.5 2271.09   338.3 2263.28
   342.5 2260.14   355.8 2256.56     530 2256.61   549.1 2260.24   558.3 2266.78
   578.4 2273.97   699.8 2269.41     714 2274.09   742.4  2274.7   767.8 2281.57
   786.1 2293.74   798.9 2304.84   818.7 2325.21   840.8 2341.02   846.3 2346.18
   868.2 2371.49   875.3 2383.79   879.2 2388.94   890.1 2408.42     910 2424.18
#Mann= 4 ,-1,0
       0      .1       0     250    .025       0   342.5    .035       0
   549.1      .1       0
Bank Sta=342.5,549.1
XS Rating Curve= 0 ,0
Exp/Cntr=0.3,0.1

Type RM Length L Ch R = 1 ,202094  ,470.6,496.9,518.5
XS GIS Cut Line= 2
2262108.70078511480113.870987594     2261185.269      480163.412
#Sta/Elev= 30
       0 2302.43   104.7 2273.69   120.7 2272.09   192.8 2271.85   228.9 2268.89
   264.9 2272.08     333 2271.94     361 2267.41   377.1 2267.32   385.1 2259.26
   401.1 2256.14   417.1 2256.09   525.3 2256.09   539.7  2259.5   561.3  2272.7
   585.4 2273.59   597.4 2281.63   645.5 2325.09   657.5 2338.55   689.5 2363.77
   717.6 2397.35     726 2413.63   733.7 2426.16   745.6    2437   813.4 2479.95
   833.7 2491.45     859 2509.07   873.8 2517.13   893.8 2522.35   924.8 2523.76
#Mann= 5 ,-1,0
       0      .1       0   385.1    .035       0   539.7      .1       0
     550     .05       0     650      .1       0
Bank Sta=385.1,539.7
XS Rating Curve= 0 ,0
Exp/Cntr=0.3,0.1

Type RM Length L Ch R = 1 ,201597  ,428.6,487.1,528.4
XS GIS Cut Line= 3
2262242.73669827479871.1684585712262021.74722683479710.873835367
     2261250.969      479558.437
#Sta/Elev= 30
       0 2314.58   112.4 2294.68     198 2272.21   230.5 2269.96   299.1 2272.14
   368.4 2269.59   466.2 2269.91     507  2263.9   515.2 2258.43   519.3  2257.8
   547.8 2255.62   653.8 2255.62   660.5 2256.34   663.9 2258.05   690.5 2271.12
   710.9  2272.2   719.1 2276.01   735.3 2292.33   751.7 2305.27   770.9 2324.47
   806.8  2356.9   854.5 2397.18   878.1 2419.49     898 2441.92   918.8  2463.5
   935.2 2478.48   948.8 2488.35     960 2495.39   975.9 2502.09  1058.7 2519.13
#Mann= 6 ,-1,0
       0      .1       0      60     .12       0     110      .1       0
   519.3    .035       0   663.9     .05       0     743      .1       0
Bank Sta=519.3,663.9
XS Rating Curve= 0 ,0
Exp/Cntr=0.3,0.1

Type RM Length L Ch R = 1 ,201110  ,510.5,533.2,548.4
XS GIS Cut Line= 2
2262379.32329331479619.947470977 2261718.5600412 479047.61087594
#Sta/Elev= 30
       0 2301.45    34.8 2296.83   126.1 2281.09     200 2272.01   252.9  2269.7
   315.8 2270.52   472.1 2267.58   486.3 2264.05   501.6 2263.09   514.6 2257.57
   538.6 2254.64   627.4 2254.56   664.9 2254.67   676.3 2257.31   676.3 2257.32
   702.7 2268.38   713.3 2269.24   718.6 2271.31   730.1  2285.3   767.9 2326.07
   782.1 2344.12   787.4 2352.09   808.5 2390.56   819.1 2402.91   835.1 2426.88
   847.3 2447.75   857.7  2473.2   863.4 2484.49   866.2 2489.13   874.2 2496.95
#Mann= 7 ,-1,0
       0      .1       0     170     .12       0     300      .1       0
   514.6    .035       0   676.3      .1       0     730     .05       0
     820      .1       0
Bank Sta=514.6,676.3
XS Rating Curve= 0 ,0
Exp/Cntr=0.3,0.1

Type RM Length L Ch R = 1 ,200577  ,556.8,562.8,567
XS GIS Cut Line= 2
2262667.24570542 479312.156473062262215.67363272  478741.1099707
#Sta/Elev= 30
       0 2288.89    41.3 2285.65    95.4 2280.13   187.4  2272.8   256.5 2270.75
   309.8  2267.7   351.7 2266.33   411.8 2266.74   420.1 2265.69     437 2261.31
   449.9 2260.35     473 2254.66   493.4 2252.91   622.2 2252.99   625.9 2253.32
     631 2254.93   636.5 2256.35   656.3 2263.93   662.1 2266.92   676.4 2269.15
   682.1 2274.88   687.1 2284.15   690.6  2289.3     695 2297.02   699.1 2306.13
   712.6 2326.06   717.7 2332.06   720.8 2334.51   722.8  2335.7     728 2336.87
#Mann= 7 ,-1,0
       0      .1       0     340     .12       0     360      .1       0
     473    .035       0     631      .1       0     670     .05       0
     720      .1       0
Bank Sta=473,631
XS Rating Curve= 0 ,0
Exp/Cntr(USF)=0,0
Exp/Cntr=0.3,0.1

Type RM Length L Ch R = 1 ,200014  ,498.3,467.8,445.4
XS GIS Cut Line= 2
2263086.72897721 478978.949902562262657.70588602478381.292633567
#Sta/Elev= 30
       0 2290.36    26.8 2288.67    41.6 2286.89    51.4 2286.25   172.2 2274.35
   238.5 2269.67   299.3 2266.33   335.6 2265.13   354.2 2265.05   415.9 2266.28
   441.6 2261.74     464 2259.32   469.9 2255.38   473.2 2253.69   477.7 2251.64
   484.5 2251.06   622.2 2250.97   642.3 2251.34     648 2253.77   659.5 2259.34
   673.8 2265.54   676.7 2266.31   685.3  2266.8   688.2 2267.92   693.9 2272.24
   706.3  2282.9   716.8  2291.1   721.1 2293.63   725.4 2294.34   735.7 2294.01
#Mann= 6 ,-1,0
       0      .1       0     400     .12       0     420    .025       0
   473.2    .035       0     648      .1       0   659.5     .05       0
Bank Sta=473.2,648
XS Rating Curve= 0 ,0
Exp/Cntr(USF)=0,0
Exp/Cntr=0.3,0.1

Type RM Length L Ch R = 1 ,199547  ,602.1,493.3,411.6
XS GIS Cut Line= 2
2263535.96283565478577.3169827622262920.12569196478044.781481695
#Sta/Elev= 30
       0 2300.22    31.1 2289.43    42.5 2286.48    70.8 2281.82   133.2 2274.53
   153.1  2272.5   184.3 2270.43   221.8 2269.91   301.1 2267.21   340.3 2265.03
   419.7 2264.11   422.8 2263.81   438.6 2258.92   453.7 2256.56   462.2 2252.78
     465 2251.38   471.1 2250.44     638 2250.48   655.4 2252.64   674.9 2256.69
   691.9 2262.63   697.8 2264.03   723.1 2265.86   750.6 2266.35   761.2  2267.2
   766.5 2269.27   774.1 2273.95   782.4 2277.12   798.2 2285.64   814.2 2291.27
#Mann= 3 ,0,0
       0      .1       0   462.2    .035       0   655.4      .1       0
Bank Sta=462.2,655.4
XS Rating Curve= 0 ,0
Exp/Cntr(USF)=0,0
Exp/Cntr=0.3,0.1

Type RM Length L Ch R = 1 ,199053  ,660.3,516.2,376.3
XS GIS Cut Line= 3
2263806.69317418477732.4003218522262976.65180659477791.901495155
2262842.77416666478000.155601718
#Sta/Elev= 30
       0 2366.05    38.6 2348.93    85.4 2331.94   146.9 2304.01     203 2283.99
   211.1 2281.73   271.2 2272.54   334.5 2266.69   351.1 2261.29   369.1 2252.95
   379.5 2250.31   535.9 2250.19   551.9 2250.22     580 2253.11   604.1 2258.01
   616.1 2262.35   628.1 2263.57   748.4  2264.4   796.4 2263.33   808.6 2261.85
   816.6 2262.93   833.1 2267.61   856.6 2265.37     874 2265.24   888.1 2267.67
   899.6 2276.14     905 2278.27   921.8 2281.22  1007.1 2289.59  1079.7 2291.01
#Mann= 3 ,-1,0
       0      .1       0   369.1    .035       0     580      .1       0
Bank Sta=369.1,580
XS Rating Curve= 0 ,0
Exp/Cntr(USF)=0,0
Exp/Cntr=0.3,0.1

Type RM Length L Ch R = 1 ,198537  ,442.4,390.3,325.7
XS GIS Cut Line= 2
2263051.02827322477205.814938116  2262839.799108 477961.47983907
#Sta/Elev= 30
       0 2378.38    40.9  2346.7    78.3 2318.83    90.7 2308.26   102.4 2297.13
   128.4    2276   144.7 2259.96   148.9 2257.37   161.3 2252.65   167.9 2251.83
   186.2 2249.91   306.7 2249.98   319.1 2251.03   323.6 2252.37   331.6 2258.64
   344.1  2260.7   367.2 2261.88   391.3 2261.35   410.8 2262.56   447.9 2261.81
   456.4 2260.44   489.4 2262.48   514.7 2266.21   522.7 2265.99   531.1 2264.65
   550.4 2264.69   586.1 2268.81   626.5 2271.34   751.1 2288.41   784.6  2290.5
#Mann= 4 ,-1,0
       0      .1       0      80    .025       0   167.9    .035       0
   323.6      .1       0
Bank Sta=167.9,323.6
XS Rating Curve= 0 ,0
Exp/Cntr(USF)=0,0
Exp/Cntr=0.3,0.1

Type RM Length L Ch R = 1 ,198147  ,474.9,446.6,416.1
XS GIS Cut Line= 2
2262524.44288949477176.0643514642262774.34781736 477961.47983907
#Sta/Elev= 30
       0 2441.25    12.3 2427.06    43.1 2398.17    61.2  2379.4    77.1 2365.02
    85.1 2356.49    97.7 2345.38   102.6 2339.38   122.9 2307.98   131.4 2297.74
   140.8 2288.96   156.5 2269.75   169.1  2258.8   180.7 2253.08   194.3 2250.37
     214 2249.41   332.8 2249.47   341.2 2250.62   345.4 2253.01   349.6 2255.84
     358 2258.69   366.4 2259.55   391.5 2259.37   408.3 2263.16   458.7 2261.91
   526.1 2266.44   605.7 2266.47     663 2268.78     749 2277.67   824.2 2288.24
#Mann= 3 ,0,0
       0      .1       0   180.7    .035       0   345.4      .1       0
Bank Sta=180.7,345.4
XS Rating Curve= 0 ,0
Exp/Cntr(USF)=0,0
Exp/Cntr=0.3,0.1

Type RM Length L Ch R = 1 ,197700  ,346,342.7,338.6
XS GIS Cut Line= 2
2262048.43350306477387.2935166922262551.21841747478107.257713664
#Sta/Elev= 30
       0 2469.08    12.1  2456.1    41.3 2412.21    67.2 2378.64    84.5 2362.91
   104.8 2339.67   118.3 2320.83     134 2293.03   138.9 2285.71   148.7 2276.52
   159.2 2262.23   164.9 2256.54   170.4 2253.59   181.2 2250.76   190.8  2247.8
   199.4 2247.62   317.2 2247.74   332.1    2251   374.6  2261.7   383.2 2262.94
   400.5 2262.21   412.1 2255.75   426.3 2254.11   432.1 2255.37   441.4 2260.64
   446.4 2262.08   607.4 2264.75   743.9 2269.78     840 2275.05   878.1  2279.9
#Mann= 5 ,-1,0
       0      .1       0     110     .08       0   181.2    .035       0
   332.1    .025       0     350      .1       0
#XS Ineff= 2 , 0
                          655.21         2279.52
Permanent Ineff=
       F       F
Bank Sta=181.2,332.1
XS Rating Curve= 0 ,0
Exp/Cntr(USF)=0,0
Exp/Cntr=0.3,0.1

Type RM Length L Ch R = 1 ,197358  ,237.8,259.2,281.8
XS GIS Cut Line= 2
2261780.67822319 477616.373033912262280.48807894478276.836057579
#Sta/Elev= 30
       0  2416.3     8.8 2413.68    14.5 2410.61    28.8 2398.06    45.6 2376.78
    51.6 2366.11    54.5 2361.87    65.5 2348.52    77.3 2332.03    86.3 2323.07
    91.3  2316.3   106.4 2291.75   111.6 2281.57   120.1 2269.46   131.4 2259.14
   148.7 2249.71     163 2246.92   276.9 2246.84   302.9 2246.94   314.3 2249.58
   332.1 2253.77   363.7 2256.86   383.6 2262.94   392.3 2262.89   407.3 2258.08
   425.7 2256.43   442.4 2260.93   562.7 2263.94     618  2266.9   828.3  2275.3
#Mann= 5 ,-1,0
       0     .08       0      70      .1       0     140    .025       0
   148.7    .035       0   314.3      .1       0
#XS Ineff= 2 , 0
                          592.68         2275.28
Permanent Ineff=
       F       F
Bank Sta=148.7,314.3
XS Rating Curve= 0 ,0
Exp/Cntr(USF)=0,0
Exp/Cntr=0.3,0.1

Type RM Length L Ch R = 1 ,197098  ,483.7,513.9,538.1
XS GIS Cut Line= 3
2261607.89712721477751.3813165082261891.47254423478295.616965324
2262154.99717418478372.955715419
#Sta/Elev= 30
       0 2349.09    20.1 2337.21    25.3  2333.6    38.1 2321.86    51.6 2311.59
    65.2 2297.87    92.2 2275.92   104.5  2264.4   111.3 2255.85   114.8 2251.35
   119.3 2248.85   132.8 2246.22   331.3 2246.22   335.8  2246.4   344.8 2248.96
   353.8 2254.28   376.4 2255.96   398.9  2262.1     408 2262.55   412.5 2261.78
   422.6 2257.45   440.4  2255.9   457.6 2261.24   556.1 2267.08   639.4 2278.42
   656.1 2279.67   700.9 2276.38   747.8 2279.45   868.7 2278.31   888.3 2279.14
#Mann= 5 ,-1,0
       0     .06       0    20.1      .1       0   111.3    .025       0
   119.3    .035       0   344.8      .1       0
Bank Sta=119.3,344.8
XS Rating Curve= 0 ,0
Exp/Cntr(USF)=0,0
Exp/Cntr=0.3,0.1

Type RM Length L Ch R = 1 ,196585  ,421.8,497.7,551.5
XS GIS Cut Line= 2
2261179.71637283477893.053489771     2261365.045      478618.178
#Sta/Elev= 30
       0 2285.74     8.4 2285.06    16.6 2282.99      29  2277.2    45.5 2267.55
    66.2 2259.03   103.3 2260.99   136.4 2259.99   160.4 2254.93   181.3 2247.76
  184.05 2246.84   194.2    2245   223.1 2244.69   355.2 2244.72   365.6 2246.87
     380 2251.77   429.5 2259.23   447.7 2259.91   466.7 2257.74     479  2261.3
   490.4  2261.7   495.6 2261.13   503.8 2257.64   507.9 2257.49   520.3 2260.39
   532.7 2261.05   681.1 2278.15   700.9 2280.95   722.6 2285.55   748.4 2293.14
#Mann= 4 ,-1,0
       0      .1       0   181.3    .025       0  184.05    .035       0
   365.6      .1       0
Bank Sta=184.05,365.6
XS Rating Curve= 0 ,0
Exp/Cntr=0.3,0.1

Type RM Length L Ch R = 1 ,196087  ,420.7,493.3,545.5
XS GIS Cut Line= 2
      2260952.87      477753.4212260597.13947471478617.349354683
#Sta/Elev= 30
       0 2268.25    21.4 2266.14      56 2267.09   103.6 2265.02   133.8 2266.65
   159.7 2265.14   177.1 2262.83   207.4 2254.96   243.5 2258.13   329.2 2258.08
   383.4 2253.28     402 2246.23     415 2244.43   553.4 2244.62   557.2 2246.03
   579.2 2259.47     601 2261.67   609.7  2264.6     627 2279.15   635.6 2284.64
   708.2 2322.15   760.3 2356.58   791.4 2379.19   804.3 2391.44   821.3 2403.86
   838.9 2423.69   843.3 2427.03   908.2 2466.24   921.1 2471.59   934.3 2474.16
#Mann= 3 ,-1,0
       0      .1       0     402    .035       0   557.2      .1       0
#XS Ineff= 2 , 0
          132.76 2277.45
Permanent Ineff=
       F       F
Bank Sta=402,557.2
XS Rating Curve= 0 ,0
Exp/Cntr=0.3,0.1

Type RM Length L Ch R = 1 ,195594  ,438.1,500,555.9
XS GIS Cut Line= 2
     2260835.517      477623.455     2260045.954      478075.883
#Sta/Elev= 30
       0 2267.37   174.4 2259.38   229.7 2253.09   285.1 2255.75     345 2255.29
   368.1 2252.87   377.3 2245.92   389.7 2244.22   506.4 2244.28   511.8    2246
     534 2257.23   552.5 2259.75   569.4 2279.77   575.2  2289.3   580.1    2300
   584.7 2306.88   619.2 2339.75   621.6 2342.99     628 2355.52   635.4 2366.58
   640.1 2372.56   649.3 2381.05   672.3 2394.85   695.4 2412.09     713 2422.83
   735.6 2439.14     808 2480.58   853.6 2512.47   865.9 2519.55     910 2552.35
#Mann= 5 ,-1,0
       0      .1       0     300    .025       0   377.3    .035       0
   511.8    .025       0     640      .1       0
Bank Sta=377.3,511.8
XS Rating Curve= 0 ,0
Exp/Cntr=0.3,0.1

Type RM Length L Ch R = 1 ,195094  ,488.5,500,516.1
BEGIN DESCRIPTION:
c/e coefficient of 0.5/0.7 to correct drawdown and capture contraction of river at this location
END DESCRIPTION:
XS GIS Cut Line= 2
     2260808.503       477452.02     2259913.239      477288.917
#Sta/Elev= 30
       0 2270.57   142.6 2259.54   276.8 2253.05   293.1 2250.71   305.3 2246.44
   337.8 2249.48   398.8 2243.69     415  2242.5   512.6  2242.5   520.8  2244.6
   549.2 2257.27   569.6 2260.24   581.7 2288.45   585.8 2293.82   614.3  2321.1
   626.5 2329.88   630.5 2333.92   640.7 2348.62   663.1 2374.72   683.4 2405.05
   687.9 2413.84   697.5 2425.78   707.8 2444.06   721.5 2458.53   745.6 2481.31
   773.1 2500.76     785 2513.58   854.2 2573.75   874.5 2587.98     910 2608.11
#Mann= 4 ,-1,0
       0      .1       0   398.8    .035       0   520.8    .025       0
   640.7      .1       0
Bank Sta=398.8,520.8
XS Rating Curve= 0 ,0
Exp/Cntr=0.7,0.5

Type RM Length L Ch R = 1 ,194594  ,513.7,500,483.2
XS GIS Cut Line= 2
     2260945.098       477046.22     2260086.091      476745.875
#Sta/Elev= 30
       0 2281.38   276.4 2253.05   296.7 2251.88   318.8 2252.35   331.5  2249.3
   353.2 2247.19   361.2 2244.79     372 2243.53   382.3 2241.49   496.8 2241.41
   560.4 2241.41   564.6 2241.83   568.8 2243.71   594.2 2257.32   611.2 2259.22
   615.4 2263.63   623.9 2285.03   632.4 2295.06   653.5 2331.72   657.7 2337.34
   691.7 2369.69   708.6 2382.99   717.4  2387.6   733.1 2399.87   755.2 2415.34
   767.6 2422.08   780.2 2426.05   827.3 2434.06   886.6 2441.11     910 2440.64
#Mann= 6 ,-1,0
       0      .1       0     290    .025       0     372    .035       0
   568.8     .12       0     600    .025       0     700      .1       0
Bank Sta=372,568.8
XS Rating Curve= 0 ,0
Exp/Cntr=0.3,0.1

Type RM Length L Ch R = 1 ,194094  ,528.5,493.2,462.5
XS GIS Cut Line= 2
     2261095.531      476511.754     2260206.281      476318.532
#Sta/Elev= 30
       0 2331.09    11.6 2326.29    36.2 2313.72    53.3 2307.26    93.5 2295.86
   142.6 2278.99     159 2272.04   183.2  2264.3   240.8 2255.98   294.1 2252.81
   347.3 2246.71   351.4 2245.63   356.6 2242.48   363.6 2239.99   515.1 2239.88
   609.2 2239.88   618.1 2242.44   633.8 2249.16   658.4 2254.44   691.1  2254.5
   699.3 2256.87   707.5 2257.75   736.1  2256.8   752.5  2264.5   760.7 2265.75
   793.4 2276.32   858.9 2289.11   879.4 2290.51   887.6 2292.38     910 2300.05
#Mann= 5 ,-1,0
       0      .1       0   356.6    .035       0   618.1      .1       0
     630    .025       0     830      .1       0
Bank Sta=356.6,618.1
XS Rating Curve= 0 ,0
Exp/Cntr=0.3,0.1

Type RM Length L Ch R = 1 ,193600  ,574.5,511.8,456.7
XS GIS Cut Line= 3
      2261162.87      475890.7312260236.62277597475965.215474738
 2259998.9489548476069.023346607
#Sta/Elev= 30
       0 2461.08    18.8 2451.52      83 2411.34    93.9 2402.89   131.1 2378.86
   159.2 2356.34   179.3 2345.03   205.3 2325.37   238.8 2302.68   283.6  2277.4
   339.8 2250.07   351.8 2241.16   355.8 2238.53   391.1 2238.48   512.3 2238.49
   536.4 2240.65   564.5 2244.03   576.6 2242.83   600.6 2247.23   659.2 2251.34
   769.2 2253.03     825 2252.09   955.9 2255.84   973.4 2254.58   986.5 2258.36
   999.6 2257.67  1060.2 2265.35  1078.4 2269.57  1130.5 2286.59  1188.6 2299.09
#Mann= 3 ,-1,0
       0      .1       0   351.8    .035       0   536.4      .1       0
Bank Sta=351.8,536.4
XS Rating Curve= 0 ,0
Exp/Cntr=0.3,0.1

Type RM Length L Ch R = 1 ,193089  ,500.2,493.6,487.4
XS GIS Cut Line= 2
     2260884.959      475184.1052259939.35365878475903.188343915
#Sta/Elev= 30
       0 2532.99    32.7 2509.13    86.4 2464.59   129.8 2434.24   153.8 2414.23
   181.9 2396.72     202 2380.42   219.8  2363.6   299.1 2300.24   357.8 2261.51
   369.6  2251.5     381 2239.73   383.8 2237.79   387.9  2237.5   510.6 2237.51
   523.6 2239.45   572.2  2242.8   578.9 2244.36   588.9 2250.01     594 2250.61
   724.6 2249.47   779.9 2251.62   960.8 2253.22   975.9 2255.37   990.9 2254.05
    1026 2255.43  1081.4 2259.41    1106  2262.9  1157.4 2271.46    1188 2280.26
#Mann= 3 ,-1,0
       0      .1       0     381    .035       0   523.6      .1       0
Bank Sta=381,523.6
XS Rating Curve= 0 ,0
Exp/Cntr=0.3,0.1

Type RM Length L Ch R = 1 ,192595  ,506.5,503.1,500.9
XS GIS Cut Line= 2
2260387.06683208474922.4257572632259699.86283208475524.908874594
#Sta/Elev= 30
       0 2370.99    41.1 2334.75    83.1    2303     106  2284.5   131.6 2265.68
   148.6 2252.03   161.9 2239.13   165.6 2236.77   168.8 2236.22   318.6 2236.26
   327.1 2238.55   338.5 2240.87   362.2 2240.23   375.3  2244.6   381.5 2248.77
   386.9  2250.6   451.9 2246.88   507.8 2250.31   579.4 2249.75   610.6 2252.84
   623.1 2252.49   631.6 2253.39   668.8 2253.81   687.1 2251.01   796.5 2252.64
   828.4 2254.51   840.2  2256.1   849.7 2259.85   860.3 2261.34   913.9 2275.72
#Mann= 4 ,-1,0
       0      .1       0     140    .025       0   161.9    .035       0
   327.1      .1       0
#XS Ineff= 2 , 0
                          660.78         2262.77
Permanent Ineff=
       F       F
Bank Sta=161.9,327.1
XS Rating Curve= 0 ,0
Exp/Cntr=0.3,0.1

Type RM Length L Ch R = 1 ,192092  ,486.5,498.6,508.1
XS GIS Cut Line= 2
2260041.94165608474549.318874594 2259405.2214774475132.076405272
#Sta/Elev= 30
       0 2325.64    15.3 2321.17    29.5 2313.01   124.2 2238.84   130.1 2235.51
   136.1 2235.03   301.3 2235.06   306.9 2235.48   315.4 2238.67   322.3    2242
   349.3 2248.36   354.9 2248.78   392.8 2248.79   414.5 2247.31   476.8 2249.35
   491.5 2247.18   510.8 2248.62   522.1 2252.75   527.1 2253.16   539.1 2252.26
   547.6 2248.07   555.5 2246.92   604.1 2248.72   663.9 2247.94   683.5 2249.42
   698.9 2251.71   710.7 2255.49   722.6  2256.8   805.2 2276.52   863.1 2291.74
#Mann= 4 ,-1,0
       0      .1       0      80    .025       0   124.2    .035       0
   315.4      .1       0
#XS Ineff= 2 , 0
                          529.58         2270.65
Permanent Ineff=
       F       F
Bank Sta=124.2,315.4
XS Rating Curve= 0 ,0
Exp/Cntr=0.3,0.1

Type RM Length L Ch R = 1 ,191593  ,468.2,501.1,529.8
XS GIS Cut Line= 3
2260051.06475726 474131.389583962259787.38891753474144.479571651
     2259186.154      474600.931
#Sta/Elev= 30
       0 2304.45      87 2298.03   135.1 2291.64   187.1  2282.2   239.2 2268.31
   283.1 2265.28   328.3 2247.05   364.4 2244.35   395.3 2247.56   438.1 2242.43
   450.4 2238.02   468.9  2233.8   639.7 2234.09   649.3  2238.1   657.9 2242.96
   675.3 2248.02   694.9 2249.13   721.6 2246.44   741.4 2251.92   754.7 2250.49
   765.2  2244.6   772.1 2242.84   795.4 2247.06   850.6  2243.2   875.7 2244.12
   889.1 2250.65   900.6 2252.97   925.9 2268.44   981.2 2294.74  1018.9 2314.88
#Mann= 6 ,-1,0
       0      .1       0     384    .025       0   450.4    .035       0
   649.3      .1       0     734     .05       0     754      .1       0
#XS Ineff= 2 , 0
                          741.63         2265.48
Permanent Ineff=
       F       F
Bank Sta=450.4,649.3
XS Rating Curve= 0 ,0
Exp/Cntr=0.3,0.1

Type RM Length L Ch R = 1 ,191092  ,463.7,504.6,541.1
XS GIS Cut Line= 3
2259954.31275188473857.9142879422259561.28445897 473793.42264916
2259018.72610925474006.279885362
#Sta/Elev= 30
       0 2286.45    46.8 2285.01    75.1  2281.5    99.5 2271.37   107.6 2265.69
   123.8 2262.35   152.1  2250.2   164.3 2248.62   184.6 2247.87   269.7 2249.31
   350.7 2246.59   468.2 2248.02   554.2 2247.06   594.8 2241.22   601.4 2237.33
   605.7 2234.54   614.3  2233.5     769 2233.68   773.3 2233.91  779.39 2237.35
   786.2 2241.18   799.1 2245.84   807.7 2245.43   821.7 2250.74   843.3 2250.03
   861.9 2257.08   934.3 2305.23   958.1 2322.93     971 2334.53   981.1 2337.66
#Mann= 7 ,-1,0
       0      .1       0  508.28     .12       0  578.28    .025       0
   601.4    .035       0  779.39      .1       0  788.28     .05       0
  898.28      .1       0
Bank Sta=601.4,779.39
XS Rating Curve= 0 ,0
Exp/Cntr=0.3,0.1

Type RM Length L Ch R = 1 ,190588  ,495.3,490.1,487.1
XS GIS Cut Line= 2
2260083.96750914473386.133824005 2258725.0976507473411.855824004
#Sta/Elev= 30
       0 2292.32    87.8 2277.98   103.8 2272.09   139.8 2252.79   159.8 2246.53
   487.9 2247.62   563.9 2244.81   651.9 2247.37   711.9 2245.46   727.9 2243.09
  737.84 2238.25   747.9 2233.25     900 2233.22   909.8 2238.41     924 2247.66
     940 2249.34     948 2255.29     976 2285.07     988 2314.56    1000 2324.78
    1012 2324.74    1080 2294.74    1100  2285.3    1132 2257.76    1148  2257.1
    1204 2273.13  1244.5 2294.25  1256.8 2296.93    1312 2320.64  1359.1    2347
#Mann= 7 ,-1,0
       0      .1       0     400     .12       0     590    .025       0
     690     .12       0  737.84    .035       0   909.8    .025       0
    1080      .1       0
Bank Sta=737.84,909.8
XS Rating Curve= 0 ,0
Exp/Cntr=0.3,0.1

Type RM Length L Ch R = 1 ,190097  ,534.5,507.7,490.7
XS GIS Cut Line= 3
2260148.00021043472858.4085306792259016.84872325472924.705518929
2258760.52976534473086.406991924
#Sta/Elev= 30
       0 2297.49    39.9 2278.37      84 2265.47   144.1 2256.89   165.2 2258.65
   236.2  2254.2   304.3  2240.7   408.5 2239.68   484.7 2244.29   628.9 2245.69
     697 2241.89   781.2  2244.7   801.2 2240.77  807.42 2236.04   817.2 2232.81
  1005.5 2232.84  1029.6 2235.71  1065.7 2242.89  1081.7 2248.29  1111.5 2249.44
  1121.7 2256.76  1129.8 2265.79    1134 2272.81  1171.7 2291.01  1190.6 2293.55
  1209.3 2309.89    1249 2328.66  1285.2 2341.18  1370.4 2363.14  1436.2 2386.65
#Mann= 5 ,-1,0
       0      .1       0  807.42    .035       0  1029.6      .1       0
    1050    .025       0 1153.09      .1       0
#XS Ineff= 2 , 0
          486.76 2262.06 1097.01         2259.12
Permanent Ineff=
       F       F
Bank Sta=807.42,1029.6
XS Rating Curve= 0 ,0
Exp/Cntr=0.3,0.1

Type RM Length L Ch R = 1 ,189590  ,556.2,502.7,465.1
XS GIS Cut Line= 3
2259550.41594403472317.5840586652258817.51979268472490.346953814
2258558.05489075472702.852754571
#Sta/Elev= 30
       0 2268.22   101.3 2259.38   117.9 2256.23   137.9 2247.23   162.6 2240.59
   183.1 2240.61   220.1  2243.8   242.3 2240.74   257.1 2235.18   265.3 2232.46
   277.2 2231.97   446.1 2232.03   457.1 2232.56   470.8 2235.23     479 2239.45
   491.3 2240.63   544.8  2240.2   610.1 2243.89   639.3 2242.81   696.8 2243.66
   721.5 2241.95   733.2 2243.01   746.5 2246.83   770.2 2246.69   804.3 2259.41
   821.9 2264.45   921.6 2279.97   949.2 2281.86   959.5 2284.96  1088.4 2305.11
#Mann= 5 ,-1,0
       0      .1       0     160     .12       0     170      .1       0
   257.1    .035       0   470.8      .1       0
Bank Sta=257.1,470.8
XS Rating Curve= 0 ,0
Exp/Cntr=0.3,0.1

Type RM Length L Ch R = 1 ,189087  ,587.7,509.7,401.7
XS GIS Cut Line= 4
     2259332.699      471695.1172258686.21572674472138.983274125
 2258477.9731776472311.9044929372258408.33836024472519.805651859
#Sta/Elev= 30
       0 2333.76    30.6 2323.06    59.4 2311.23    95.5 2299.13   146.2 2284.57
   180.2 2275.41   223.4 2267.01   307.5 2247.24   354.8 2243.42   367.2 2234.71
     373 2231.63   378.7 2230.85   516.8 2230.91   553.8 2234.87   571.5 2238.92
   585.9 2237.91     612 2240.51   659.7 2240.79   698.1 2238.08   718.7 2240.52
   741.2 2240.54     781 2243.56   869.6 2242.44   944.2 2239.59   963.3 2245.44
   988.9 2247.19  1005.2 2254.23  1028.6 2257.83  1161.7 2270.47  1274.1 2287.39
#Mann= 5 ,-1,0
       0      .1       0     280     .12       0     300    .025       0
   367.2    .035       0   553.8      .1       0
Bank Sta=367.2,553.8
XS Rating Curve= 0 ,0
Exp/Cntr=0.3,0.1

Type RM Length L Ch R = 1 ,188577  ,501.1,479,452
XS GIS Cut Line= 3
2258584.33770667471260.4158213122258531.91416082472035.162978042
2258367.07812271472488.215215817
#Sta/Elev= 30
       0 2553.36    52.9 2516.24      93  2476.3   133.1  2443.1   161.1 2416.35
   165.1 2411.99   177.2 2391.86   194.2 2376.99   213.2 2356.02   225.3 2348.53
   254.4 2323.02   277.4 2298.97  356.57 2231.94   369.6 2229.81   489.9  2229.9
   505.9 2231.25     558 2230.66   578.1 2237.16   602.1 2235.06   634.2 2238.99
   670.3 2238.08   686.3 2241.35   722.4 2242.47   838.3 2242.34   937.1 2239.38
   962.9 2245.74     983 2246.47  1059.6 2258.96  1187.3 2272.81  1258.6  2283.4
#Mann= 4 ,-1,0
       0      .1       0     310    .025       0  356.57    .035       0
   505.9      .1       0
Bank Sta=356.57,505.9
XS Rating Curve= 0 ,0
Exp/Cntr=0.3,0.1

Type RM Length L Ch R = 1 ,188098  ,503.6,504.6,505.3
XS GIS Cut Line= 3
2258030.99776265471390.3526399332258148.13159302472118.464620667
     2258160.581472439.364690522
#Sta/Elev= 30
       0 2451.87      14 2444.77    31.2 2431.99    63.6 2395.47    87.9 2371.97
   115.2 2347.39   124.4 2337.55   132.6 2326.56   144.7 2315.42   167.5 2290.75
   177.1 2281.94   201.4  2254.8   209.5  2239.3   213.5 2235.41   219.9 2231.55
   233.8 2228.69   399.9 2228.74   416.1 2231.13   448.5 2239.92   468.8 2241.21
   558.4 2238.61   626.8  2238.5   683.5 2242.19   699.7 2239.78   707.8 2240.86
     724 2246.53   763.3 2246.68   784.2 2249.64   900.3 2259.49  1058.6 2279.61
#Mann= 4 ,-1,0
       0      .1       0     190    .025       0   219.9    .035       0
   416.1      .1       0
Bank Sta=219.9,416.1
XS Rating Curve= 0 ,0
Exp/Cntr=0.3,0.1
