HEC-RAS study GRNBRRRV.prj: GRNBRRRV

--- GRNBRRRV.g01 (geometry) --- (continued)

Type RM Length L Ch R = 1 ,161093  ,532.9,490.4,446.4
XS GIS Cut Line= 3
     2251826.822      463878.0012251060.28297425 464180.28440819
 2250589.7212914464247.599186383
#Sta/Elev= 30
       0 2439.46    58.7 2409.48   123.2 2362.52   220.4 2290.09   299.5 2232.97
     319 2211.28   333.9 2198.29     353 2195.02   371.5 2182.12   380.7 2179.25
   497.3 2179.25     536 2181.94   540.3 2182.88   553.2 2189.65   570.4 2192.74
   609.1 2189.32   695.6  2187.9   798.3 2191.47   863.8 2190.24   874.4 2190.09
   896.8 2190.42   927.4 2197.76   949.4 2191.56   969.6 2189.75  1151.4 2189.75
  1199.9 2193.51  1223.9 2203.29    1254  2220.8  1280.7 2239.04  1299.3 2255.58
#Mann= 10 ,-1,0
       0      .1       0   123.2     .12       0   220.4      .1       0
   371.5    .035       0     536    .025       0   540.3     .05       0
   863.8    .025       0   874.4     .05       0  1151.4      .1       0
    1254     .05       0
#XS Ineff= 2 , 0
       0                   927.4       0    2210
Permanent Ineff=
       F       F
Bank Sta=371.5,536
XS Rating Curve= 0 ,0
Exp/Cntr=0.3,0.1

Type RM Length L Ch R = 1 ,160603  ,477.4,470.5,463.4
XS GIS Cut Line= 3
     2251445.941       463322.252250942.47065111463829.524991566
2250572.62667051463992.746739181
#Sta/Elev= 30
       0 2425.42     9.8 2420.46    87.7 2369.66    94.3 2366.87   147.6 2326.27
   178.7  2308.1   201.2 2292.08   229.6 2274.43   249.4 2258.47     289 2233.43
   325.8 2198.41   348.4 2194.72   370.4 2181.13   377.3 2178.78   530.6 2178.81
   546.4 2181.04   567.7 2186.93   584.6 2189.24   628.4 2186.69   689.6 2190.02
   769.7 2188.61     803 2195.04   817.8 2190.61   830.9 2189.75     971 2189.75
   992.7 2191.31  1014.5 2197.97  1040.8 2212.66  1083.2 2240.83    1119  2259.7
#Mann= 8 ,-1,0
       0      .1       0     110     .12       0     170    .025       0
   370.4    .035       0   546.4      .1       0     590     .05       0
  724.71    .025       0  944.71      .1       0
Bank Sta=370.4,546.4
XS Rating Curve= 0 ,0
Exp/Cntr=0.3,0.1

Type RM Length L Ch R = 1 ,160132  ,543.2,514.2,477.5
XS GIS Cut Line= 2
2251095.24374892 462963.023131752250373.07591873463795.086066535
#Sta/Elev= 30
       0 2420.56    34.9 2414.12    71.8  2402.8      84 2395.86   119.4 2381.34
     167 2357.01   193.9 2337.28   247.6 2289.79   254.9 2281.66   262.4 2276.94
   329.8 2224.91   358.1 2199.72   366.6 2195.14   386.5 2193.98   407.4 2182.38
     416 2178.16   553.7 2178.06   590.5 2178.12     602 2182.31   611.9 2183.75
   627.5  2182.1   664.4 2186.76   818.5 2185.64   865.1 2187.01   882.1 2192.44
     894 2199.33   964.9 2227.61  1004.6 2241.31  1048.2 2251.68  1101.8 2259.57
#Mann= 9 ,-1,0
       0      .1       0     190     .12       0     250    .025       0
   407.4    .035       0     602     .05       0     840      .1       0
     850     .05       0     970      .1       0    1000     .05       0
Bank Sta=407.4,602
XS Rating Curve= 0 ,0
Exp/Cntr(USF)=0,0
Exp/Cntr=0.3,0.1

Type RM Length L Ch R = 1 ,159618  ,539.7,505.4,463.9
XS GIS Cut Line= 2
2250535.30202551462633.3378179672250082.63885659463609.311008768
#Sta/Elev= 30
       0 2424.86     8.6 2422.36    35.1 2409.08    43.9 2402.49    57.1 2396.59
    83.6 2375.05   101.2 2368.74   145.3 2358.72   207.1 2324.19   219.1 2316.87
   237.2 2302.75   291.4 2256.12   330.5 2218.11   352.6 2199.62   361.4 2194.28
   383.4 2192.93   402.9 2179.68   414.3 2176.72   586.3 2176.72   596.9 2179.26
   608.3 2182.28   625.8 2181.13     648 2186.09     689 2183.59   837.6 2192.83
   868.5 2196.63     930 2209.49   981.2 2216.72  1043.7 2234.97  1075.8 2237.39
#Mann= 7 ,-1,0
       0      .1       0     200     .12       0     230    .025       0
   402.9    .035       0   596.9      .1       0     690     .05       0
     930      .1       0
Bank Sta=402.9,596.9
XS Rating Curve= 0 ,0
Exp/Cntr(USF)=0,0
Exp/Cntr=0.3,0.1

Type RM Length L Ch R = 1 ,159112  ,560,541.1,516.9
XS GIS Cut Line= 2
2249899.48034893462455.4124105292249771.26939357463598.844808331
#Sta/Elev= 30
       0 2461.16      34 2468.37    54.1 2468.54    62.2 2465.98    78.3 2451.51
    82.3 2449.35   102.4 2448.85   106.4 2446.63   114.5 2439.25   130.6 2421.07
   154.7 2391.12   219.1 2330.33   255.4 2303.74   344.8 2216.34     364 2195.15
   368.1 2192.75   380.1 2192.48   384.2 2191.13   406.3 2178.84   406.3  2178.8
   412.3 2175.57   585.4 2175.58   601.5 2178.92   641.8 2184.13     686 2184.13
   728.4 2187.53   810.8 2189.54   859.1 2192.93  1084.5 2220.07  1150.6 2229.36
#Mann= 6 ,-1,0
       0      .1       0     260     .12       0     360    .025       0
   406.3    .035       0   601.5      .1       0     660     .05       0
Bank Sta=406.3,601.5
XS Rating Curve= 0 ,0
Exp/Cntr(USF)=0,0
Exp/Cntr=0.3,0.1

Type RM Length L Ch R = 1 ,158571  ,481.3,462.8,439.3
XS GIS Cut Line= 2
2249271.50832268462518.2096131542249357.85447629463630.243409643
#Sta/Elev= 30
       0 2472.91       7 2468.79      19  2456.3   115.1 2392.64   135.4 2376.02
   148.6 2362.82   159.4 2349.24   185.2 2320.02   223.6 2273.43   235.7 2263.97
   251.7 2248.67   259.7 2238.41   283.8  2215.4   291.8 2204.93   295.9 2200.76
   311.9 2191.07     328 2190.22     336 2183.36   348.22177.107     356  2174.6
   508.5 2174.11   525.32176.661   540.6 2179.34   580.7 2183.54   600.8 2183.12
   644.9 2186.17   728.9 2188.01   901.7 2200.15  1066.2 2214.68  1115.4 2217.36
#Mann= 5 ,-1,0
       0      .1       0     300    .025       0   348.2    .035       0
   525.3      .1       0     690     .05       0
Bank Sta=348.2,525.3
XS Rating Curve= 0 ,0
Exp/Cntr(USF)=0,0
Exp/Cntr=0.3,0.1

Type RM Length L Ch R = 1 ,158108  ,542.4,515.4,488.7
XS GIS Cut Line= 2
 2248719.4162496462549.6082144662249036.01881283463700.890262597
#Sta/Elev= 30
       0 2457.42    32.7 2452.52    61.8 2445.41   103.3 2422.61   144.8 2392.78
   218.3  2335.5   244.3 2309.03   260.6 2295.92   270.3 2285.56   281.7 2275.58
   289.9 2266.47   306.5 2252.83   319.1  2239.9   335.6 2226.48   348.4 2209.74
   364.6 2191.91   385.4 2188.27   410.2 2175.51   422.7 2173.69   582.7 2173.72
  593.982175.765   601.1 2179.02     612 2179.78   630.1 2184.29   667.5 2183.19
   803.9 2187.55     895  2196.1  1011.8 2199.92  1078.2 2204.38    1194 2217.28
#Mann= 5 ,-1,0
       0      .1       0     190    .025       0   410.2    .035       0
  593.98     .05       0    1190      .1       0
Bank Sta=410.2,593.98
XS Rating Curve= 0 ,0
Exp/Cntr(USF)=0,0
Exp/Cntr=0.3,0.1

Type RM Length L Ch R = 1 ,157593  ,514.3,502.3,492.3
XS GIS Cut Line= 2
     2248151.012        462829.62248692.89661488463779.445284462
#Sta/Elev= 30
       0 2271.97    26.9 2270.57    73.9 2276.89   117.8 2286.58   155.7 2293.29
   192.9 2297.14   211.7  2296.3   220.6 2292.24   229.8 2284.41   252.7 2255.43
   270.3 2236.99   276.8 2228.37   293.8 2212.01   312.7 2191.99   317.2 2188.76
   334.8  2186.4   358.7 2174.37   364.1 2172.17   372.5 2171.34   515.3 2171.38
   528.4 2174.01   538.3 2177.77   561.3 2183.27   570.6 2184.19   616.3  2181.6
   651.5 2184.99   736.9 2184.73   879.1 2193.84  1011.4 2198.14  1093.5 2205.46
#Mann= 6 ,-1,0
       0      .1       0     210     .12       0     260    .025       0
   358.7    .035       0   528.4     .05       0     550      .1       0
#XS Ineff= 2 , 0
                          774.19         2212.85
Permanent Ineff=
       F       F
Bank Sta=358.7,528.4
XS Rating Curve= 0 ,0
Exp/Cntr=0.3,0.1

Type RM Length L Ch R = 1 ,157091  ,474.7,494.8,515.4
XS GIS Cut Line= 2
     2247694.808      463135.6342248336.06264566464027.509606345
#Sta/Elev= 30
       0 2245.35    70.9 2245.88     154 2242.47   189.1 2240.49   233.5 2234.17
   265.8 2227.73   285.8 2220.43     303 2211.73   331.2 2188.15     346 2186.38
   372.4 2174.17   386.1  2170.1     518 2170.02   532.3 2170.73   540.9 2174.07
   568.5 2181.55   691.6 2183.97   716.3 2191.67     731 2189.77   810.9 2189.81
   831.4 2193.21     869 2193.43   903.5 2204.42   918.2 2203.84   947.8 2198.65
   992.1 2199.55  1041.4 2203.82  1070.2 2212.14  1090.7 2212.06  1098.5 2214.59
#Mann= 8 ,-1,0
       0     .05       0     210    .025       0     330      .1       0
   372.4    .035       0   540.9    .025       0     570      .1       0
     690    .025       0     810      .1       0
Bank Sta=372.4,540.9
XS Rating Curve= 0 ,0
Exp/Cntr=0.3,0.1

Type RM Length L Ch R = 1 ,156596  ,463.6,505.1,558.8
XS GIS Cut Line= 3
2247464.97553434463407.0293727652247464.32956565463604.610556478
     2247721.692      464161.868
#Sta/Elev= 30
       0 2236.99    70.2    2233   102.2 2230.13   110.2 2228.55   114.2 2227.43
   122.2 2223.19   126.2 2219.46   134.5 2206.56   142.2 2199.81   149.8 2194.92
   170.2 2188.36   186.2 2187.58     207 2185.03   220.2 2181.32   233.5 2180.62
   251.1 2174.34   268.7 2171.84   281.9 2169.81   440.5 2169.84   449.3 2171.71
   460.1 2177.79   478.2 2179.84     489 2182.96   559.7 2182.72   636.1 2184.73
   678.5 2187.15   718.1 2191.48   757.8 2198.32     793 2209.59   811.4 2217.31
#Mann= 4 ,-1,0
       0    .025       0   268.7    .035       0   449.3    .025       0
  497.58      .1       0
Bank Sta=268.7,449.3
XS Rating Curve= 0 ,0
Exp/Cntr=0.3,0.1

Type RM Length L Ch R = 1 ,156091  ,431.4,482.8,543.6
XS GIS Cut Line= 3
 2247243.2154599 463366.869416042247049.30888186 463701.00245723
     2247064.211      464356.958
#Sta/Elev= 30
       0 2231.87     7.3 2231.04    27.3 2224.09    82.9 2194.63   106.3 2187.05
     146 2184.22     183  2186.3   196.9 2182.32   348.7 2184.39   444.1 2182.93
   462.5 2180.53   486.5 2173.23   510.6 2171.03   530.5 2169.53   694.7  2169.6
     707 2171.23   734.6 2185.46   810.6 2184.46   834.6 2188.99   854.6 2201.86
   870.6 2209.78   886.6  2215.5   906.6 2220.19   922.6 2228.76   950.6 2238.74
   981.3 2258.97   998.7 2265.89  1014.7 2275.92  1030.7 2286.98  1042.4 2298.44
#Mann= 5 ,-1,0
       0      .1       0     100     .05       0     380    .025       0
   510.6    .035       0     707      .1       0
Bank Sta=510.6,707
XS Rating Curve= 0 ,0
Exp/Cntr=0.3,0.1

Type RM Length L Ch R = 1 ,155608  ,472.4,512.9,550.4
XS GIS Cut Line= 2
 2247003.7200127463038.3218193832246371.11118638464204.882869591
#Sta/Elev= 30
       0 2225.75    21.5 2222.64    75.5  2199.3    96.2 2192.27     108 2190.01
   184.7 2187.86   200.4 2186.09   259.2 2185.59   279.1 2182.68   317.2 2180.79
   421.9 2180.81   490.1 2182.69   565.3 2180.52   644.9 2182.91   726.7 2182.58
   745.3 2181.64   758.6 2175.71   795.4 2171.86     813 2169.29   922.4 2169.29
   945.9 2171.86   954.3 2173.26   969.5 2180.14  1004.3 2200.01  1027.1 2207.69
  1077.1 2230.25  1163.6 2273.88  1184.9 2289.03  1240.9 2335.04    1327  2399.4
#Mann= 6 ,-1,0
       0      .1       0      80     .05       0     750    .025       0
   795.4    .035       0   945.9    .025       0     980      .1       0
Bank Sta=795.4,945.9
XS Rating Curve= 0 ,0
Exp/Cntr=0.3,0.1

Type RM Length L Ch R = 1 ,155095  ,477.2,504.1,534.4
XS GIS Cut Line= 2
2246923.04562782 462909.24450894     2245846.799       463750.91
#Sta/Elev= 30
       0 2226.18    13.8 2220.84    59.5 2195.75    84.3 2185.64      96 2183.96
   150.2 2182.88     210 2184.53   220.7 2183.12   399.7  2179.4   512.1 2181.27
   566.2 2178.86     626 2181.08   771.4 2181.75   788.5 2176.11   808.4 2175.82
   834.1 2170.67   846.6    2169   973.7 2169.01   983.7 2170.75   993.4 2172.83
   998.9 2175.79    1004 2183.02  1009.1 2192.81  1014.2 2198.17  1075.1 2207.85
  1104.8 2220.82  1155.7 2249.77  1187.4 2274.21  1227.4 2310.35  1366.3 2428.81
#Mann= 8 ,-1,0
       0      .1       0     160     .05       0     320     .03       0
     480     .05       0     790    .025       0     800      .1       0
   834.1    .035       0   983.7      .1       0
Bank Sta=834.1,983.7
XS Rating Curve= 0 ,0
Exp/Cntr=0.3,0.1

Type RM Length L Ch R = 1 ,154591  ,486.4,500.3,516.2
XS GIS Cut Line= 2
2246777.54544779462673.762645698     2245515.502      463234.123
#Sta/Elev= 30
       0  2214.8    64.2  2190.5    94.6 2187.48   145.9 2182.81   176.6 2183.81
   224.7 2181.12   255.3 2182.46   312.2 2181.82   424.9 2178.21   526.7 2179.26
   621.9 2178.12   732.4  2180.5   797.7 2181.55   830.4 2171.01   846.2 2168.72
    1030 2168.72  1034.4 2168.91  1038.7 2171.18  1051.9 2180.17  1060.6 2182.15
  1073.5 2194.16  1128.1 2238.15  1165.7 2261.47    1170 2269.08  1176.7 2283.69
  1181.4 2291.12  1231.1 2344.77  1310.5 2423.66  1337.2 2446.29  1380.9 2479.87
#Mann= 5 ,-1,0
       0      .1       0    94.6     .05       0   732.4    .025       0
   830.4    .035       0  1038.7      .1       0
#XS Ineff= 2 , 0
       0   164.3    2190               0
Permanent Ineff=
       F       F
Bank Sta=830.4,1038.7
XS Rating Curve= 0 ,0
Exp/Cntr=0.3,0.1

Type RM Length L Ch R = 1 ,154091  ,514.5,496.3,481.2
XS GIS Cut Line= 2
2246571.27652222462329.738229658     2245343.706      462706.912
#Sta/Elev= 30
       0  2243.7    57.6 2203.31    78.6 2191.25    99.5 2183.28   107.9 2181.97
   141.3 2183.37   158.9 2180.11   183.2 2179.41     292 2179.91   342.2 2177.82
     380 2178.41   492.8 2178.53   529.2 2176.55   622.6 2176.69   635.1 2175.27
   690.3 2177.86   714.6 2174.97   731.4 2170.79   748.1 2168.19   911.6 2168.16
   927.1 2170.55   936.4 2173.97   944.8  2179.8   953.1 2182.07   971.9 2201.19
  1049.4 2264.31  1116.3 2326.55    1200  2398.5  1225.1 2415.36  1284.2 2448.37
#Mann= 8 ,-1,0
       0      .1       0   183.2     .05       0     292     .07       0
     380     .05       0   492.8     .07       0   690.3    .025       0
   731.4    .035       0   927.1      .1       0
#XS Ineff= 2 , 0
       0   124.6    2190               0
Permanent Ineff=
       F       F
Bank Sta=731.4,927.1
XS Rating Curve= 0 ,0
Exp/Cntr=0.3,0.1

Type RM Length L Ch R = 1 ,153595  ,511,496.8,486
XS GIS Cut Line= 2
2246405.00505021461752.319173685       2245191.9      462293.622
#Sta/Elev= 30
       0 2242.87    22.5 2229.17    49.1  2216.3    86.1 2205.17   136.7 2185.98
   154.2 2181.05   184.9  2181.1     198 2176.61   249.6 2175.48   491.5 2178.58
   671.1 2178.72     693 2177.57   725.1  2173.4   736.8 2169.13   745.5 2167.49
   968.9 2167.47   982.6  2169.3    1004 2177.55  1012.9  2177.8    1022 2179.72
  1060.9 2180.32  1091.6 2182.99  1104.7 2185.24  1113.5 2188.76  1152.9  2210.3
    1223 2255.59  1258.2 2280.27    1288 2303.86  1297.9 2310.64  1328.4 2335.37
#Mann= 5 ,-1,0
       0      .1       0     180     .05       0     650    .025       0
   736.8    .035       0   982.6      .1       0
Bank Sta=736.8,982.6
XS Rating Curve= 0 ,0
Exp/Cntr=0.3,0.1

Type RM Length L Ch R = 1 ,153098  ,496.8,507.3,512.4
XS GIS Cut Line= 2
2246245.97497577461196.031800919     2244995.722      461877.014
#Sta/Elev= 30
       0 2249.86    25.8 2241.74    52.2 2230.57    61.3 2225.78    69.3 2218.13
    74.9 2214.59    88.6 2211.43   127.8  2193.2   161.5 2182.22   188.8 2179.58
   225.2 2179.73   235.1 2175.51   243.5 2174.41   298.1 2174.55   373.7 2178.23
   479.9 2178.62   565.4 2175.36   721.6 2178.19   785.5 2177.56   807.2 2167.67
   812.8 2166.53   879.1 2166.53  1086.1 2167.63    1123  2178.8  1267.2 2178.33
  1323.7 2180.46  1340.4 2185.18  1357.1 2194.25  1382.2 2209.93  1423.7  2239.7
#Mann= 6 ,-1,0
       0      .1       0   161.5     .05       0   721.6     .08       0
   807.2     .07       0   879.1    .035       0  1086.1      .1       0
Bank Sta=807.2,1086.1
XS Rating Curve= 0 ,0
Exp/Cntr=0.3,0.1

Type RM Length L Ch R = 1 ,152590  ,431.6,498.4,544
XS GIS Cut Line= 2
2246067.65000693460783.043484128     2244712.765      461427.744
#Sta/Elev= 30
       0 2258.36    16.2 2252.47    34.9 2240.54   105.7  2189.2   127.9 2175.89
   158.9 2173.47   167.7 2173.78   172.5 2176.35   190.3  2178.6   207.6 2173.71
   234.2 2176.23   318.4 2172.42   721.5 2176.88     831 2174.12   849.9 2175.88
   863.2 2172.33   876.5 2172.48   885.4 2166.48   979.5 2165.05  1147.8 2166.19
  1155.6 2168.78  1164.4 2175.54  1173.3 2178.44  1288.5    2177  1350.5 2178.43
  1399.2 2184.93  1423.9 2192.34  1439.5 2199.37    1475 2222.78  1500.5 2242.69
#Mann= 8 ,-1,0
       0      .1       0   172.5     .05       0   721.5     .08       0
     831    .025       0   885.4     .08       0   979.5    .035       0
  1147.8    .025       0  1164.4      .1       0
Bank Sta=885.4,1147.8
XS Rating Curve= 0 ,0
Exp/Cntr=0.3,0.1

Type RM Length L Ch R = 1 ,152092  ,529.5,476.7,428.4
XS GIS Cut Line= 3
2245937.90190621460452.2808545612245295.99366633460730.782212933
      2244564.56      460781.526
#Sta/Elev= 30
       0 2253.89    41.1 2250.93      75 2240.16   102.2 2224.98   119.6 2212.27
   150.1  2182.5   160.1 2179.21   180.7 2178.29   193.7 2173.43   372.5 2174.63
   385.2 2172.48   490.2 2175.28   546.9 2173.91   779.7 2175.75   795.8 2175.22
   823.8 2170.26     833 2165.85   843.9 2163.75  1076.4 2163.75  1084.7 2165.93
  1108.5 2174.12  1185.5 2174.39  1220.8  2170.7  1252.9 2175.73  1308.8 2188.65
  1333.1 2200.25  1353.1 2213.65  1409.2 2258.48  1425.3 2269.62  1432.9 2277.13
#Mann= 6 ,-1,0
       0      .1       0     240     .05       0     670     .08       0
  779.72    .025       0     833    .035       0  1084.7      .1       0
Bank Sta=833,1084.7
XS Rating Curve= 0 ,0
Exp/Cntr=0.3,0.1

Type RM Length L Ch R = 1 ,151615  ,470.5,522,583.7
XS GIS Cut Line= 3
2245758.50831738460056.8272856312245196.44234519460161.277657404
     2244474.972       460481.55
#Sta/Elev= 30
       0 2218.63    29.8 2211.85    88.1 2194.37   111.4 2186.95   128.5 2178.84
   148.8 2177.93     157 2174.72   177.3 2171.72   300.8 2174.16     336 2170.66
   364.5 2169.74   527.2 2174.28   742.7 2173.96   750.6 2172.88   764.5 2167.53
   792.8 2164.15   799.6 2162.87   847.7 2162.84  1028.9 2162.93  1040.3  2164.5
  1066.5 2166.63    1084 2170.23  1127.8 2194.16  1140.9 2204.51  1158.4 2221.42
  1180.3 2239.99  1215.3 2263.99    1272 2306.54  1342.2 2363.93  1361.1 2377.19
#Mann= 7 ,-1,0
       0      .1       0     150     .05       0  651.69      .1       0
  761.69    .025       0   792.8    .035       0  1040.3    .025       0
 1081.69      .1       0
Bank Sta=792.8,1040.3
XS Rating Curve= 0 ,0
Exp/Cntr=0.3,0.1

Type RM Length L Ch R = 1 ,151093  ,504.4,498.1,492.3
XS GIS Cut Line= 2
  2245698.058367      459782.503     2244389.104      459781.519
#Sta/Elev= 30
       0 2225.32    25.9 2222.61    45.9 2212.83   113.9 2174.23   133.9 2171.69
   169.9 2176.05   205.9 2170.47   305.9 2174.01   404.9 2174.86   529.9 2169.21
   598.8 2172.82   693.9 2173.36   717.9 2169.34   762.6  2167.9   789.2 2163.83
   801.9    2162   933.9    2162   941.9 2164.12   970.5 2184.17   989.9 2201.68
  1005.9 2209.43  1021.9 2220.46  1033.9 2233.44  1057.9 2254.73  1117.9 2299.55
  1129.4 2304.09  1150.3 2320.14  1237.9 2374.94  1269.5 2392.13    1309  2410.3
#Mann= 6 ,-1,0
       0      .1       0      80     .05       0     670     .08       0
     770    .025       0   789.2    .035       0   941.9      .1       0
Bank Sta=789.2,941.9
XS Rating Curve= 0 ,0
Exp/Cntr=0.3,0.1

Type RM Length L Ch R = 1 ,150595  ,501.2,499.9,500
XS GIS Cut Line= 2
 2245693.4958142459241.901683208     2244388.495      459306.149
#Sta/Elev= 30
       0 2197.62    21.3 2195.02    33.4 2189.04    61.4 2179.35    81.4 2178.07
    93.4 2175.19   133.5 2173.03   265.6 2168.66   273.7 2169.75   285.7 2175.97
   297.7 2176.81   301.7 2176.45   317.7 2167.62   509.9 2174.16     570 2173.32
   671.9 2172.76   702.2 2168.24   746.2  2166.1   760.1 2163.05   766.2 2161.38
   942.5 2161.38   949.9  2163.2   954.5 2167.69   970.5 2201.41   978.5 2209.48
   994.5 2220.11  1059.4 2256.98  1111.3 2283.36  1134.7  2292.9  1306.6 2321.89
#Mann= 9 ,-1,0
       0     .06       0      80      .1       0     180     .05       0
     570      .1       0     670    .025       0   760.1    .035       0
   949.9      .1       0    1060     .05       0    1260      .1       0
Bank Sta=760.1,949.9
XS Rating Curve= 0 ,0
Exp/Cntr=0.3,0.1

Type RM Length L Ch R = 1 ,150095  ,528.8,500.3,480.3
XS GIS Cut Line= 3
2245588.53969857458617.9539344652245026.87800909458774.200122393
     2244362.021       458806.85
#Sta/Elev= 30
       0 2226.58    91.7 2173.65    95.9 2172.54   131.4 2169.92   282.7 2171.57
   299.3 2169.17   307.6 2169.88   321.2  2175.3   332.5 2176.34     344 2175.34
   357.4 2170.74   382.4 2173.39   432.2 2171.65   473.9 2161.84     482 2164.96
   515.2 2166.42   540.1  2170.8     565 2172.25   629.7 2171.18   653.8 2168.07
   665.8 2163.77   677.8 2160.76   874.7 2160.79   888.4 2164.61     907 2172.86
   934.1 2180.29  1014.2 2220.68  1050.3 2236.86  1110.3 2246.75  1248.6  2261.5
#Mann= 6 ,-1,0
       0     .06       0      80      .1       0  582.99    .025       0
   665.8    .035       0   888.4      .1       0  982.99     .05       0
Bank Sta=665.8,888.4
XS Rating Curve= 0 ,0
Exp/Cntr=0.3,0.1

Type RM Length L Ch R = 1 ,149595  ,522.1,500,485.2
XS GIS Cut Line= 2
2245388.19258716458147.261228046     2244301.196      458388.227
#Sta/Elev= 30
       0 2221.32    49.2 2196.16      82 2176.33   110.6 2170.81   225.4 2169.17
   237.7 2174.09   245.8 2175.22     254 2174.89   266.3 2169.55   274.5 2169.01
   368.8 2171.79   450.7 2171.63   487.6 2168.75   495.8 2163.41     504 2160.04
   632.1 2160.03   749.8 2160.06   753.9 2160.29   759.6 2163.89   770.3 2168.59
   819.9 2171.71   839.9 2175.98   848.1 2179.53   872.7 2198.01     885 2205.26
   901.4 2211.36   920.5 2215.09   979.2 2220.38  1028.4 2218.04  1113.4 2225.66
#Mann= 11 ,-1,0
       0      .1       0      70     .06       0     170      .1       0
     270     .06       0     370      .1       0     470    .025       0
   495.8    .035       0   759.6    .025       0     780     .05       0
     980     .06       0    1080     .05       0
Bank Sta=495.8,759.6
XS Rating Curve= 0 ,0
Exp/Cntr=0.3,0.1

Type RM Length L Ch R = 1 ,149095  ,519.5,500.7,488.9
XS GIS Cut Line= 2
2245153.26517956457616.011296198     2244176.516      457962.714
#Sta/Elev= 30
       0 2215.59    26.6 2202.97    52.1 2192.78    69.1 2189.81    90.3 2183.13
    98.8 2178.01   111.5 2175.44   158.2 2174.18   170.9 2170.66   187.9 2169.15
   264.3 2169.12   350.3 2172.27   378.9 2171.93   412.1 2167.47   418.4 2162.89
   421.5 2160.39   429.9 2159.16   667.5 2159.16   671.8  2159.6   677.6 2162.93
   684.5 2166.49   697.3 2166.72   709.7 2170.33   718.5 2171.27   838.2 2171.73
   879.8 2175.19   934.9 2190.82   964.7 2195.27   985.9    2200  1036.5 2205.73
#Mann= 8 ,-1,0
       0      .1       0      30     .06       0     230      .1       0
     350    .025       0   418.4    .035       0   677.6     .05       0
     820     .06       0     970     .05       0
Bank Sta=418.4,677.6
XS Rating Curve= 0 ,0
Exp/Cntr=0.3,0.1

Type RM Length L Ch R = 1 ,148594  ,500.4,501.3,502.3
XS GIS Cut Line= 2
2244929.06745217457101.913478373     2243981.699      457553.162
#Sta/Elev= 30
       0 2197.98    18.7    2186    24.1 2183.44    36.4 2173.91    54.1 2172.84
      63 2168.51    71.9 2166.71   132.2 2167.68   159.2 2166.52   226.9 2166.71
   311.1 2169.38   390.9 2173.23   417.3 2170.58   429.3 2166.26   435.5 2162.25
   441.3 2159.34   448.5 2158.56   665.6 2158.56     670 2159.27   674.4 2161.74
   696.6 2167.37   714.4 2167.69   753.4 2170.47   861.4 2169.29   906.5  2170.4
   957.5 2173.01  1002.3 2194.41    1020 2201.71  1026.5  2203.7  1049.3 2207.96
#Mann= 7 ,-1,0
       0     .05       0     330     .06       0   435.5    .035       0
   674.4    .025       0     690     .05       0     920     .06       0
     980     .05       0
Bank Sta=435.5,674.4
XS Rating Curve= 0 ,0
Exp/Cntr=0.3,0.1

Type RM Length L Ch R = 1 ,148093  ,402.9,455.8,508
XS GIS Cut Line= 4
2244899.48424848456616.9477682922244826.28799951456606.441542057
2244557.30076792 456726.71686545      2243770.49      457095.332
#Sta/Elev= 30
       0 2233.16    35.7 2225.31    59.9 2217.13    98.2 2192.51   106.9 2188.09
   124.5 2173.35     142 2172.11   155.1 2165.49   159.4 2164.86   198.9 2165.16
   276.6 2168.83   416.4 2168.97   602.9 2172.15   612.8 2169.65     629 2168.52
     642 2161.28   648.1 2158.43   652.5 2158.19   877.8 2158.23   885.7 2161.55
   891.1 2166.12   894.7 2166.76   930.7 2164.22   972.9 2164.05  1045.1 2167.84
  1087.2 2164.55  1123.3 2168.33  1147.4 2179.69  1195.5 2207.28  1237.5  2228.1
#Mann= 8 ,-1,0
       0      .1       0  283.95     .05       0   558.6     .06       0
   618.6    .025       0     642    .035       0   885.7     .05       0
  1048.6     .06       0  1158.6      .1       0
Bank Sta=642,885.7
XS Rating Curve= 0 ,0
Exp/Cntr=0.3,0.1

Type RM Length L Ch R = 1 ,147637  ,525.3,543.4,568.8
XS GIS Cut Line= 5
2244917.37490187 456389.87955835  2244800.409603456341.568542504
2244171.71679371 456466.393749192243883.76573514456473.745961117
     2243608.129      456408.958
#Sta/Elev= 30
       0 2220.54   113.8 2209.29   143.1 2205.08   151.3 2202.38   167.6 2194.02
   179.8 2182.49     192 2174.07   200.2 2171.61   228.5 2171.53     241 2165.56
   245.1 2164.93   285.8 2164.35   493.9 2169.53   738.5 2170.44   754.8 2169.17
783.64242159.927   795.1 2157.91   987.1 2157.88991.53082159.821   999.1  2164.8
  1011.1 2163.94  1031.2 2166.24  1071.6 2200.87  1079.8 2212.56  1095.6 2228.62
  1182.5  2309.6  1215.4 2334.86  1256.5 2369.11  1308.5 2415.87  1338.7 2438.93
#Mann= 9 ,-1,0
       0      .1       0  196.55     .06       0  296.55     .07       0
  396.55     .05       0  486.55     .06       0  706.55    .025       0
783.6424    .035       0991.5308     .06       0  997.51      .1       0
Bank Sta=783.6424,991.5308
XS Rating Curve= 0 ,0
Exp/Cntr=0.3,0.1

Type RM Length L Ch R = 1 ,147094  ,528.6,504.4,488.7
XS GIS Cut Line= 2
2245290.42444705456084.726253969     2243729.956       455882.59
#Sta/Elev= 30
       0  2240.6    74.9 2224.06   300.7 2190.19   365.3 2195.97   421.7  2190.5
   530.6 2190.21   551.5 2184.39   583.1 2169.68   627.4  2163.9   651.6  2164.9
   671.8 2171.49   708.1 2163.75   739.9 2166.78   796.9 2162.95   990.5 2169.74
  1002.6 2168.82  1014.7 2161.49  1026.4 2157.53  1184.1 2157.47  1194.3 2162.22
  1208.3 2171.86  1244.6 2174.89    1282 2216.36  1321.2 2254.37  1337.3 2284.98
  1341.4 2289.47  1409.9 2347.52  1470.4 2393.18  1510.8 2413.29  1573.5 2424.33
#Mann= 8 ,-1,0
       0      .1       0     270     .05       0     470      .1       0
     860     .07       0     960    .025       0  1014.7    .035       0
  1194.3     .06       0    1260      .1       0
Bank Sta=1014.7,1194.3
XS Rating Curve= 0 ,0
Exp/Cntr=0.3,0.1

Type RM Length L Ch R = 1 ,146589  ,533.3,495.2,469.8
XS GIS Cut Line= 3
2245303.26071733454637.7945144952244745.71692706455398.312841575
     2243751.172      455471.109
#Sta/Elev= 30
       0 2256.76    41.8 2232.64   108.4 2203.66   133.4 2183.61   143.1 2179.75
   343.5 2179.16   420.8 2173.72   480.3 2177.12     557 2176.46   812.6 2169.05
   860.3 2171.08  1165.1  2164.5  1213.3 2169.71  1233.3 2161.45  1273.4 2168.16
  1293.5  2167.1  1313.7 2159.36  1337.6 2159.31  1369.7 2163.87  1385.7 2159.64
  1409.8 2157.12  1526.1 2157.12  1534.1 2159.65  1550.2  2169.5  1578.2 2195.63
  1602.3 2198.68  1642.2 2251.54  1674.5 2266.56  1718.6 2274.34  1940.2 2289.81
#Mann= 5 ,-1,0
       0      .1       0  1385.7    .035       0  1534.1      .1       0
    1553     .06       0    1653      .1       0
#XS Ineff= 2 , 0
          845.07 2190.45
Permanent Ineff=
       F       F
Bank Sta=1385.7,1534.1
XS Rating Curve= 0 ,0
Exp/Cntr=0.3,0.1

Type RM Length L Ch R = 1 ,146094  ,428,416.7,405
XS GIS Cut Line= 3
2244538.10722674454598.4109580552244343.85656739454854.732173388
     2243668.555      455132.343
#Sta/Elev= 30
       0 2195.63      76 2176.86    91.9 2167.64    97.6 2166.02   118.9 2166.75
   159.1 2164.12   188.9 2166.79     246  2165.8   269.5 2162.13   294.6 2165.06
   307.8 2168.78   317.4 2168.86   329.9 2168.08   347.8 2161.79   459.7 2164.58
   479.6 2161.67   491.8 2157.68   498.6 2156.16   658.6 2156.19   672.6 2157.65
   703.3 2161.06   723.5 2167.79   753.7 2168.01   776.8 2171.76   810.6 2181.16
   840.2 2187.26   938.2 2191.89   966.9 2190.87   987.3 2194.56  1051.7 2201.16
#Mann= 8 ,-1,0
       0      .1       0  441.61    .025       0   491.8    .035       0
   672.6    .025       0  761.61      .1       0  791.61     .06       0
  861.61     .05       0 1051.61     .06       0
#XS Ineff= 2 , 0
          312.87 2184.22
Permanent Ineff=
       F       F
Bank Sta=491.8,672.6
XS Rating Curve= 0 ,0
Exp/Cntr=0.3,0.1

Type RM Length L Ch R = 1 ,145678  ,330.8,283.1,226.1
XS GIS Cut Line= 3
2244415.33379936454311.2867353852243685.60704663454706.676529692
2243618.73965494455134.046380892
#Sta/Elev= 30
       0  2302.7   117.3 2261.53   167.4 2247.37   180.8 2242.27   194.7 2235.98
   248.6 2205.47   285.7 2187.82     313 2170.09     349 2168.81     363 2161.59
   372.1 2159.74   390.3 2160.91   399.4 2159.24   426.7 2163.06   458.5  2163.9
   472.2 2162.58   481.7 2156.97   485.8 2155.53   499.4 2155.34     636 2155.35
     647 2156.75   676.9  2158.8   694.2 2157.62   756.1 2166.11   945.9 2166.13
   974.2 2167.74  1061.6 2182.46    1124 2188.59    1173 2190.82  1262.5 2199.32
#Mann= 8 ,-1,0
       0      .1       0     430    .025       0   481.7    .035       0
     647      .1       0     690     .05       0 1069.96     .06       0
 1169.96      .1       0 1259.96     .06       0
Bank Sta=481.7,647
XS Rating Curve= 0 ,0
Exp/Cntr(USF)=0,0
Exp/Cntr=0.3,0.1

Type RM Length L Ch R = 1 ,145394  ,336.2,282.7,224
XS GIS Cut Line= 3
2243967.98977381454011.1029485252243622.62419746454571.416331134
2243588.81218299455151.050864868
#Sta/Elev= 30
       0 2358.44      87 2301.32   105.8 2294.18     181 2249.68     199 2235.41
   213.1 2226.03   228.1 2211.29   242.7 2199.85   256.2 2185.66   265.9 2167.52
   303.2 2167.88   319.8 2161.48   329.9  2155.9   335.7 2154.66   467.6 2154.48
   487.92156.166   528.7 2159.56   542.8 2159.41   563.8  2155.1   585.1 2157.43
   627.4 2165.75   670.2  2164.7     708 2166.28   908.3 2166.59   942.6 2171.44
  1004.6 2182.91  1120.7 2189.08    1196 2195.65  1220.9    2198  1238.8 2202.07
#Mann= 5 ,-1,0
       0      .1       0   329.9    .035       0   487.9     .08       0
   670.2     .05       0    1196      .1       0
Bank Sta=329.9,487.9
XS Rating Curve= 0 ,0
Exp/Cntr(USF)=0,0
Exp/Cntr=0.3,0.1

Type RM Length L Ch R = 1 ,145112  ,496.6,488.7,479.8
XS GIS Cut Line= 2
2243473.37575998454008.9298338562243540.24315166 455186.37738308
#Sta/Elev= 30
       0 2342.41    52.3 2299.56    84.4 2269.77    96.4 2256.53   136.5 2221.82
   152.5 2203.09   168.5 2174.68   172.5  2169.5   176.5 2168.15   192.6 2167.38
   208.82156.069   216.6 2153.94   328.8    2154   340.12155.971   424.9 2161.68
     449 2159.97   464.5 2163.46     485 2165.63   637.3 2166.28   692.9 2164.62
   765.5 2165.51   785.5 2167.04   845.6 2178.96   881.7 2182.64   965.8 2184.28
    1086 2192.38  1134.1 2197.66  1150.1 2201.29  1166.1 2200.82  1179.3 2205.38
#Mann= 9 ,-1,0
       0      .1       0     140    .025       0   208.8    .035       0
   340.1      .1       0     440     .05       0     830     .06       0
     930     .05       0    1030      .1       0    1130     .06       0
Bank Sta=208.8,340.1
XS Rating Curve= 0 ,0
Exp/Cntr(USF)=0,0
Exp/Cntr=0.3,0.1

Type RM Length L Ch R = 1 ,144623  ,523,520.3,523
XS GIS Cut Line= 2
 2242955.8802939 454035.095334952243156.48246895455285.224831656
#Sta/Elev= 30
       0    2316    22.4 2307.35    57.9 2285.55    83.1  2275.1   135.8 2264.73
   152.2 2258.61   168.2  2245.9   183.6 2228.05   192.5 2216.41   204.8 2194.62
   224.9 2171.81     233 2165.02   253.3 2163.71   267.4 2155.26   277.6 2152.84
   407.2 2152.88   415.3  2155.7   423.4  2160.8   431.5 2162.59   565.2 2163.73
   646.2 2162.37   824.5 2170.32   969.1 2179.19  1116.2 2192.92  1147.1 2198.59
  1168.8  2205.1  1189.1 2205.94  1197.2 2210.83    1210 2214.29  1266.1 2233.96
#Mann= 7 ,-1,0
       0      .1       0     120    .025       0   267.4    .035       0
   415.3      .1       0     420     .05       0    1120     .06       0
    1210      .1       0
Bank Sta=267.4,415.3
XS Rating Curve= 0 ,0
Exp/Cntr(USF)=0,0
Exp/Cntr=0.3,0.1

Type RM Length L Ch R = 1 ,144103  ,376.7,380.6,385.3
XS GIS Cut Line= 3
2242483.72238532454043.0862726082242462.38546642454279.223366031
2242673.95733985455372.300662663
#Sta/Elev= 30
       0 2233.82    77.9  2220.4   110.5 2216.04   186.9 2208.64     223 2203.07
     288 2174.49   300.2 2167.96   304.3 2166.61   324.7 2166.06   353.5 2154.38
   361.3 2151.75   573.2 2151.78   577.3 2151.98   583.3 2154.09   638.4 2161.09
   707.6  2163.4   817.6 2164.98   875.2  2167.2   972.5 2167.77  1013.2 2166.85
  1073.2  2169.4  1114.2 2172.72  1175.6 2178.83  1196.5  2183.6  1225.1 2184.81
  1265.8 2194.76  1282.1  2202.6  1302.5 2203.12  1322.8  2214.8  1350.5 2226.68
#Mann= 7 ,-1,0
       0      .1       0   307.1    .025       0   353.5    .035       0
   583.3      .1       0   707.1     .05       0  1207.1     .07       0
  1307.1     .06       0
#XS Ineff= 2 , 0
                          873.13         2177.56
Permanent Ineff=
       F       F
Bank Sta=353.5,583.3
XS Rating Curve= 0 ,0
Exp/Cntr=0.3,0.1

Type RM Length L Ch R = 1 ,143722  ,456.4,469.7,480.9
XS GIS Cut Line= 4
2242071.85913369454087.3017955442242089.25338253454307.682592768
2242155.65824491454725.0845849172242504.13619239455385.701864632
#Sta/Elev= 30
       0 2189.71      42 2182.18   190.5 2169.64   206.5 2168.06   214.5 2165.72
   233.8 2165.92     255 2164.49   271.2 2162.04   323.8 2162.64   344.1 2156.94
   350.72152.686   356.2 2150.97   587.1 2151.07  593.072152.587   615.5  2158.9
   631.7 2159.77   712.3 2159.72   789.2 2161.75   943.2 2163.23  1023.7 2165.06
  1037.3 2166.24  1136.8 2167.38  1177.5 2169.61  1236.3 2170.75    1260 2174.16
  1286.6 2175.09  1335.8 2188.09  1363.6 2197.68  1381.4 2205.31  1390.6  2205.8
#Mann= 9 ,-1,0
       0      .1       0   350.7    .035       0  593.07    .025       0
  663.72     .05       0  993.72     .06       0 1103.72     .05       0
 1223.72     .07       0 1323.72     .05       0 1333.72     .06       0
#XS Ineff= 2 , 0
                          802.14         2174.05
Permanent Ineff=
       F       F
Bank Sta=350.7,593.07
XS Rating Curve= 0 ,0
Exp/Cntr=0.3,0.1

Type RM Length L Ch R = 1 ,143252  ,313.1,316,318
XS GIS Cut Line= 3
2241863.63087239454011.2616894152241649.90539273454396.896794008
2241705.65986569455209.982857908
#Sta/Elev= 30
       0 2187.77    31.9 2184.67    70.8 2176.26   162.8 2172.46   180.5 2164.56
   212.6  2166.7   221.7 2171.69   226.3 2171.98   248.2 2169.53   279.4 2161.21
   315.9 2159.61   441.2 2162.33   493.3 2161.03   522.1 2153.56   544.6 2151.47
   553.4 2149.84     751 2149.56     766 2149.67   769.7 2151.48     778 2158.89
     790 2161.87   926.3 2161.52   946.4 2163.04   958.4 2166.11   998.5 2164.57
  1030.6 2171.55  1070.7 2184.16  1102.7 2198.29  1110.8 2199.28  1255.9 2276.62
#Mann= 7 ,-1,0
       0      .1       0     180     .05       0     390      .1       0
   544.6    .035       0   769.7      .1       0   890.9     .05       0
  1080.9      .1       0
Bank Sta=544.6,769.7
XS Rating Curve= 0 ,0
Exp/Cntr(USF)=0,0
Exp/Cntr=0.3,0.1

Type RM Length L Ch R = 1 ,142936  ,316.7,349.9,391.3
XS GIS Cut Line= 4
2241835.75363591453964.7996286212241352.54820365454448.005060881
2241361.84061581454940.5029053012241515.16541643455098.473912001
#Sta/Elev= 30
       0 2196.27    22.6 2196.64    50.9 2193.33    96.7 2180.31   119.3 2176.75
   155.5 2174.44   175.9 2176.04   200.8 2165.25   226.8 2165.82   243.2 2172.41
   251.7 2173.36   257.4 2172.09   271.5 2164.14   294.7 2160.57   725.7 2160.57
   788.5 2156.03   800.6 2152.11   820.6 2150.58   844.6 2148.97   988.6 2148.94
   996.72150.574  1012.6 2156.36  1032.6 2159.79  1080.5 2158.53  1132.6 2163.31
  1149.8 2169.34  1175.9 2182.07  1260.1 2203.57  1316.7  2221.8  1396.1 2252.26
#Mann= 5 ,-1,0
       0      .1       0     260     .05       0     640      .1       0
   820.6    .035       0   996.7      .1       0
Bank Sta=820.6,996.7
XS Rating Curve= 0 ,0
Exp/Cntr(USF)=0,0
Exp/Cntr=0.3,0.1

Type RM Length L Ch R = 1 ,142587  ,465.8,512,570.7
XS GIS Cut Line= 3
2241699.54101815453811.9467265722241137.45035498454310.844729072
      2240851.42      455059.787
#Sta/Elev= 30
       0 2187.34   134.4 2170.33   198.8 2164.16   221.4 2165.17   298.7 2159.95
   598.4  2160.5     657 2158.97   792.6 2160.86   822.5 2157.69   852.5 2159.57
     869 2157.61   942.5 2158.71   998.1 2156.76  1032.4 2154.191045.199 2150.72
  1070.9 2148.52  1165.1 2148.441196.7992151.068  1207.9 2157.58  1220.8 2175.09
  1259.7 2210.54  1268.7 2222.14  1302.1 2256.85  1323.5 2276.42  1387.8 2327.71
    1405 2338.06  1417.4 2344.84  1429.8 2349.17  1447.7 2352.61  1553.3 2356.65
#Mann= 6 ,-1,0
       0      .1       0     290     .05       0     690      .1       0
 1001.56    .025       01045.199    .035       01196.799      .1       0
Bank Sta=1045.199,1196.799
XS Rating Curve= 0 ,0
Exp/Cntr=0.3,0.1

Type RM Length L Ch R = 1 ,142075  ,483.2,483.8,486.9
XS GIS Cut Line= 2
2241509.62780155453679.087932005     2240243.748      454601.625
#Sta/Elev= 30
       0 2199.99    31.2  2197.2    54.1 2191.92   105.4 2168.69   120.6 2165.35
     140 2163.87   173.3 2165.61   214.6  2159.9   674.9 2158.28   827.1 2159.87
   864.3 2154.57   922.4 2159.22   991.7 2159.89  1007.5 2158.49  1029.1 2150.99
  1046.1 2149.25  1070.4 2147.72  1169.9 2147.76  1176.4 2149.34    1185 2154.02
  1204.5 2179.26  1219.2 2194.02  1293.6 2241.55  1313.8 2251.66  1338.2 2258.61
    1358 2257.51  1409.4 2247.75  1521.3 2220.46  1554.3 2204.69  1566.4 2200.58
#Mann= 7 ,-1,0
       0      .1       0     280     .05       0     800      .1       0
     970    .025       0    1010      .1       0  1046.1    .035       0
  1176.4      .1       0
Bank Sta=1046.1,1176.4
XS Rating Curve= 0 ,0
Exp/Cntr=0.3,0.1

Type RM Length L Ch R = 1 ,141591  ,464.5,489,513.8
XS GIS Cut Line= 2
2241266.30270382453303.641273467     2239966.273      454187.254
#Sta/Elev= 30
       0 2203.66    52.5 2199.71   100.5 2191.45   123.6 2183.37   133.2 2176.75
   145.1  2172.8     161 2162.83   176.7 2163.32   191.2 2160.42   264.7 2155.58
   636.2 2157.91   873.1 2156.64   950.5 2158.87   989.2 2155.311010.5742149.793
  1033.5 2146.98  1192.3 2147.031203.4742150.333    1212 2156.25  1226.6 2169.76
  1269.6 2198.65  1308.4 2227.72  1318.5 2241.11  1342.3  2261.6  1361.8 2275.14
  1397.4 2296.51  1447.2 2315.56  1476.9  2337.1  1511.4  2359.5  1571.9 2391.37
#Mann= 6 ,-1,0
       0      .1       0     280     .05       0     810      .1       0
     930    .025       01010.574    .035       01203.474      .1       0
#XS Ineff= 2 , 0
          231.33 2181.22
Permanent Ineff=
       F       F
Bank Sta=1010.574,1203.474
XS Rating Curve= 0 ,0
Exp/Cntr=0.3,0.1

Type RM Length L Ch R = 1 ,141102  ,665.1,699.1,735.5
XS GIS Cut Line= 3
2241064.67482309453070.3511413762240492.37454893453352.717428912
     2239672.281      453679.586
#Sta/Elev= 30
       0 2194.77    31.8  2188.6    83.1 2165.95     110 2164.51   116.5 2162.49
   143.3  2161.8     179 2153.48   250.3 2152.34   325.1  2154.6   575.9 2156.22
   716.5  2155.1   926.9 2158.34   952.7    2154   969.9 2152.98   978.6  2148.8
  1004.4 2146.06  1150.8 2146.071163.7622149.039  1168.8 2152.01  1186.7 2172.08
  1211.3 2193.27  1223.7 2201.98    1336 2305.73  1348.9 2311.72  1366.1  2329.2
    1379 2338.36  1417.6 2370.39  1447.9 2393.48  1465.1 2404.62    1521 2447.61
#Mann= 7 ,-1,0
       0     .12       0      80      .1       0     190     .05       0
  848.17      .1       0  948.17    .025       0   978.6    .035       0
1163.762      .1       0
Bank Sta=978.6,1163.762
XS Rating Curve= 0 ,0
Exp/Cntr=0.3,0.1

Type RM Length L Ch R = 1 ,140403  ,300.9,312.1,326.6
XS GIS Cut Line= 3
 2241115.5916936452701.031575017 2240641.6786735452780.017078367
2239633.45195426452845.063963479
#Sta/Elev= 30
       0  2199.8    64.3 2194.92   128.2 2186.95   180.4 2182.56   258.9 2171.03
   315.7 2167.64   319.8  2166.8   327.9 2162.05   348.2 2160.89   364.6 2153.02
   380.6 2150.51   437.4 2150.12     486 2153.27   710.4 2155.03   890.8 2153.67
   958.9 2155.86   995.1 2152.52  1032.42146.252  1039.1 2144.78  1203.5 2144.84
  1213.4 2146.25    1221 2150.31  1247.5  2175.9  1291.6 2213.48  1331.7 2255.57
  1343.7 2264.86    1372 2298.39  1403.9 2328.12  1423.9 2344.75  1490.8  2394.7
#Mann= 8 ,-1,0
       0      .1       0     230     .12       0     330      .1       0
     430     .05       0  920.45      .1       0 1020.45    .025       0
  1032.4    .035       0  1213.4      .1       0
Bank Sta=1032.4,1213.4
XS Rating Curve= 0 ,0
Exp/Cntr(USF)=0,0
Exp/Cntr=0.3,0.1

Type RM Length L Ch R = 1 ,140091  ,470.7,492.7,518.1
XS GIS Cut Line= 3
2240844.97673075452474.5209684922240428.77060938452529.688248655
     2239578.306       452485.08
#Sta/Elev= 30
       0 2201.91    33.1 2199.52    61.3 2194.81   113.5 2173.39   131.3 2161.66
   154.1 2159.77     167 2152.16   178.3 2149.96   242.9 2150.09   263.1 2152.19
   516.6  2154.2   592.7    2152   672.8 2155.39   696.8 2151.69   720.9 2150.64
736.6763 2146.57   748.9 2144.25   913.1 2144.28927.47352147.088  1001.2  2207.7
  1028.7 2233.55  1049.3 2253.56  1065.3  2272.4  1077.3 2284.05  1085.4 2296.25
  1104.7 2317.43  1113.4 2325.65  1225.5 2416.46  1245.6 2430.64  1271.5 2451.13
#Mann= 7 ,-1,0
       0     .12       0      50      .1       0     150     .05       0
  549.85      .1       0  649.85    .025       0736.6763    .035       0
927.4735      .1       0
Bank Sta=736.6763,927.4735
XS Rating Curve= 0 ,0
Exp/Cntr=0.3,0.1

Type RM Length L Ch R = 1 ,139598  ,481.9,511.3,536.5
XS GIS Cut Line= 2
2240795.45922281452202.080066844     2239675.798      451908.917
#Sta/Elev= 30
       0 2197.02    28.2 2194.24    44.7 2190.54    65.7 2183.32   102.6 2167.37
   119.2 2162.72     144 2158.95   168.8 2159.95   201.9 2151.11   210.1 2150.01
   370.4 2149.97   536.8 2153.24     574 2150.85   594.7 2145.82   598.8 2143.65
   602.9 2143.41   784.9 2143.44   798.7 2146.03   805.6 2149.46   825.9  2165.1
   842.8 2181.09   846.9 2186.45   855.2 2205.69   859.3 2211.59   863.4 2215.28
   929.6 2269.21   958.5 2295.22    1034 2358.73    1075 2391.05  1157.4 2459.49
#Mann= 6 ,-1,0
       0     .12       0     110      .1       0     210     .05       0
     490      .1       0   594.7    .035       0   798.7      .1       0
Bank Sta=594.7,798.7
XS Rating Curve= 0 ,0
Exp/Cntr=0.3,0.1

Type RM Length L Ch R = 1 ,139087  ,467.3,482.8,495.5
XS GIS Cut Line= 2
2240820.63258847451828.7895897792239993.36742989451384.732112715
#Sta/Elev= 30
       0 2188.31    23.7 2185.08    64.1  2175.5    86.8 2169.57     114 2158.55
   132.2 2158.03   150.3  2155.8     260  2155.7     325 2153.84   372.8 2148.31
   390.9 2148.23     450 2151.43   481.6 2148.32   499.3 2144.29   504.4 2142.55
     509 2142.53   667.9 2142.53     677 2144.18   695.1 2157.68   709.6 2172.19
   713.3 2177.01   727.3 2202.73   731.4 2208.69   745.1 2222.44   760.4 2250.63
     774 2268.09   847.9 2336.36   862.7 2351.38   883.3    2375   938.9 2425.18
#Mann= 5 ,-1,0
       0      .1       0     140     .05       0     260      .1       0
   499.3    .035       0     677      .1       0
Bank Sta=499.3,677
XS Rating Curve= 0 ,0
Exp/Cntr=0.3,0.1

Type RM Length L Ch R = 1 ,138604  ,372.7,376.2,379.3
XS GIS Cut Line= 2
2241147.30863916451565.5148189982240199.93434105450887.305030645
#Sta/Elev= 30
       0 2198.69    71.3    2196   110.5 2192.46   203.2 2177.04   263.4 2162.81
     299 2157.84   343.3 2157.88   426.6 2154.29   461.2 2154.62   540.1 2148.78
   591.5 2147.47   607.4 2148.72   623.7 2146.03     6322143.013   646.5 2141.06
   800.8 2141.08   813.8 2143.01   819.6 2146.81   835.2 2162.28     850 2172.85
   893.9 2219.11   935.1 2258.42   958.2 2276.87     973 2301.76   985.8 2315.67
  1037.5 2356.23  1080.5 2394.06  1100.9 2419.32  1114.9 2433.14  1165.1 2488.11
#Mann= 4 ,-1,0
       0      .1       0     560     .07       0     632    .035       0
   813.8      .1       0
Bank Sta=632,813.8
XS Rating Curve= 0 ,0
Exp/Cntr(USF)=0,0
Exp/Cntr=0.3,0.1

Type RM Length L Ch R = 1 ,138228  ,341.6,317.7,293.3
XS GIS Cut Line= 2
 2241437.6672048451340.8578266062240505.12874581450630.856954424
#Sta/Elev= 30
       0 2221.05    82.3 2206.53   380.5 2167.77   514.6 2160.97   524.7 2159.02
   531.7 2155.54   549.9 2155.83   594.5  2152.2   610.2 2148.91     643 2148.76
   655.4 2146.25   685.9  2147.6   710.7 2145.56   725.8 2142.09   735.9 2140.28
   886.7 2140.28   899.22142.152   904.1 2144.79   915.4 2155.27   952.1 2180.38
   965.6 2191.78   979.8 2212.82   987.2 2220.97   997.3 2237.14  1002.3  2243.5
  1047.6 2284.41    1094 2323.92    1123 2353.74  1165.4 2393.71  1172.1 2402.06
#Mann= 3 ,-1,0
       0      .1       0   725.8    .035       0   899.2      .1       0
Bank Sta=725.8,899.2
XS Rating Curve= 0 ,0
Exp/Cntr(USF)=0,0
Exp/Cntr=0.3,0.1

Type RM Length L Ch R = 1 ,137910  ,309.9,316.4,326.1
BEGIN DESCRIPTION:
mannings n increased in this area to correct drawdown and is more representative of imagery
END DESCRIPTION:
XS GIS Cut Line= 3
2241619.93608542450669.0062550192241265.99535212 450713.51377238
2240628.05426995450429.513423507
#Sta/Elev= 30
       0  2205.8    56.2 2192.39   116.7 2183.82   148.9 2181.46   248.5 2178.88
   261.4 2177.26   294.1 2169.15   393.7 2163.97   450.7 2158.88   468.2 2154.03
   490.1 2154.56   564.5 2146.37   586.4 2148.68   625.8 2144.56   635.9 2141.66
   647.7 2139.72   779.5 2139.75   792.2 2141.27   797.7 2143.48   815.8 2156.97
   844.7  2174.9   898.5 2213.49   910.4 2229.44   919.2 2237.46   932.3 2246.66
   949.8 2269.94   962.9 2285.01  1006.7 2322.76    1033 2364.08    1055 2384.05
#Mann= 3 ,-1,0
       0      .1       0   635.9     .04       0   792.2      .1       0
#XS Ineff= 2 , 0
          484.06 2168.59
Permanent Ineff=
       F       F
Bank Sta=635.9,792.2
XS Rating Curve= 0 ,0
Exp/Cntr(USF)=0,0
Exp/Cntr=0.3,0.1

Type RM Length L Ch R = 1 ,137594  ,511.9,505.7,497.8
XS GIS Cut Line= 2
     2241504.135      450514.409     2240705.316      450078.532
#Sta/Elev= 30
       0 2184.78    13.6 2183.08    45.5 2183.52    95.6 2180.96   180.7 2173.59
   227.8 2166.63   250.6 2159.73   259.7 2154.84   264.2 2153.89     287 2153.34
   304.5 2150.58   345.8 2146.66   359.9 2146.73   381.2 2140.38   387.3 2139.22
   560.4 2139.22   566.9 2139.97   575.8 2143.24   587.8 2152.82   619.7  2152.6
   628.7 2156.03   642.5 2163.08   715.4 2213.92   751.8 2244.21   773.3 2260.54
   792.8 2271.18   820.4 2281.05   842.9  2286.9   874.8 2292.02     910 2295.07
#Mann= 4 ,-1,0
       0      .1       0     360    .025       0   381.2    .035       0
   566.9      .1       0
Bank Sta=381.2,566.9
XS Rating Curve= 0 ,0
Exp/Cntr=0.3,0.1

Type RM Length L Ch R = 1 ,137088  ,594.2,489.1,371.8
XS GIS Cut Line= 3
     2241732.795      450033.2142241189.27034338449777.728069461
     2240865.269       449742.72
#Sta/Elev= 30
       0 2240.81    27.2 2231.77      36 2230.43    53.7 2224.34    72.7 2220.07
   138.8 2199.58   208.4 2181.01   239.4 2171.19   280.1 2162.15     288 2160.04
   296.8 2154.38   301.2 2153.03   327.8 2152.51   345.4 2143.04   355.3 2139.33
   548.7 2138.31   557.6 2139.18   588.5 2150.12   601.7 2146.84   625.8 2146.68
   686.2 2149.83   734.4 2149.49   782.7 2146.86   798.8 2142.47   801.8 2143.08
     823 2155.06     835 2167.45   859.2 2183.26   887.3 2195.73   926.5 2207.69
#Mann= 6 ,-1,0
       0      .1       0   280.1    .025       0   355.3    .035       0
   557.6     .05       0   601.7    .025       0   801.8      .1       0
#XS Ineff= 2 , 0
                           686.2         2165.03
Permanent Ineff=
       F       F
Bank Sta=355.3,557.6
XS Rating Curve= 0 ,0
Exp/Cntr=0.3,0.1

Type RM Length L Ch R = 1 ,136599  ,541.5,505.2,466.2
XS GIS Cut Line= 2
     2241623.106      449113.1022240851.21827261449667.260794235
#Sta/Elev= 30
       0 2359.82    13.6 2350.17      43 2336.13   144.2 2274.84   162.7 2265.94
   211.4 2238.86     240 2226.88   269.5 2212.43     304 2189.94   329.4  2169.2
   343.2 2155.85   353.2 2151.74   374.8 2149.62   387.7 2141.32   394.8 2138.32
   486.6 2137.56   521.4 2138.27   540.3 2144.36   561.1 2146.31   589.6 2147.53
   717.6 2147.99   742.2 2149.54   801.3 2147.52   835.8 2141.93   860.4 2149.38
     885 2164.34   899.8 2176.57   907.9 2181.89   932.9 2193.16   950.2 2199.12
#Mann= 7 ,-1,0
       0      .1       0     370    .025       0   394.8    .035       0
   521.4      .1       0     540     .05       0     660    .025       0
     780      .1       0
#XS Ineff= 2 , 0
                          738.02         2161.39
Permanent Ineff=
       F       F
Bank Sta=394.8,521.4
XS Rating Curve= 0 ,0
Exp/Cntr=0.3,0.1

Type RM Length L Ch R = 1 ,136094  ,511.9,500,489.9
XS GIS Cut Line= 2
     2241089.045      448666.354      2240647.57      449462.093
#Sta/Elev= 30
       0 2361.69    35.1 2343.15    53.5 2330.83    67.4 2323.01    94.7 2304.02
   129.2  2284.2   183.2 2245.11     191 2241.65   214.5 2225.64   264.6  2198.8
   305.1 2174.09   323.4 2162.04   337.2 2149.63   341.7 2148.26     360 2147.26
   381.1 2137.96   387.5  2136.2   506.4 2136.18   517.6 2137.81   541.1 2138.66
   561.3 2146.22   570.7 2147.86   611.6 2146.94   652.8 2140.39   675.7 2145.36
   761.8 2147.48   780.9 2151.68   806.5 2159.43   873.6 2185.84     910 2195.71
#Mann= 5 ,-1,0
       0      .1       0     310    .025       0   381.1    .035       0
   517.6    .025       0     530      .1       0
Bank Sta=381.1,517.6
XS Rating Curve= 0 ,0
Exp/Cntr=0.3,0.1
