HEC-RAS study GRNBRRRV.prj: GRNBRRRV

--- GRNBRRRV.g01 (geometry) --- (continued)

Type RM Length L Ch R = 1 ,135594  ,514.1,500,488.5
XS GIS Cut Line= 2
     2240580.999      448443.454     2240239.297      449286.864
#Sta/Elev= 30
       0 2379.75     6.2 2374.51    19.1    2366      45  2346.1    83.9 2318.29
   112.5 2300.96   131.3  2291.5   178.8 2262.73   183.2 2258.58   196.1 2250.97
   217.7 2234.15   238.5 2216.18   247.9 2205.39   312.2 2158.76   321.2 2150.94
   325.5 2148.82   343.1  2147.3   364.4 2136.69   368.7 2135.17   377.3 2135.06
   524.1 2135.06   532.7 2136.73   545.6  2139.4     564 2141.31   674.6 2147.62
   723.7 2151.93   778.7 2154.95   826.2 2162.35   860.7 2171.92     910  2181.7
#Mann= 6 ,-1,0
       0      .1       0     320    .025       0   364.4    .035       0
   532.7     .05       0     740     .06       0     850      .1       0
Bank Sta=364.4,532.7
XS Rating Curve= 0 ,0
Exp/Cntr=0.3,0.1

Type RM Length L Ch R = 1 ,135094  ,510.2,500,491.9
XS GIS Cut Line= 2
     2240055.767      448274.209     2239813.067      449151.248
#Sta/Elev= 30
       0 2389.36    36.3 2363.92    69.5 2338.08    73.5 2334.01    81.9 2321.32
    90.2  2312.2   102.9 2303.36   115.1 2291.51   131.7 2277.94   177.4 2251.67
   185.7 2248.05   210.1 2230.44   264.6 2198.51   281.2 2183.11   297.8 2154.21
   301.9 2149.89   322.7  2145.8   340.2 2136.26   347.6 2134.06   530.2 2134.11
   538.4 2135.91   559.2 2142.53     580 2144.93     663  2145.7   756.3 2152.14
   770.9 2154.72   787.5 2155.06   799.9 2157.57   849.7  2162.4     910 2175.57
#Mann= 7 ,-1,0
       0      .1       0     280    .025       0   340.2    .035       0
   538.4      .1       0     580     .05       0     690     .06       0
     890      .1       0
Bank Sta=340.2,538.4
XS Rating Curve= 0 ,0
Exp/Cntr=0.3,0.1

Type RM Length L Ch R = 1 ,134594  ,505.3,500,495.5
XS GIS Cut Line= 2
     2239533.913      448157.916     2239359.315       449051.01
#Sta/Elev= 30
       0 2355.87    35.9 2336.15    72.4 2310.77   113.4 2284.03   154.1 2254.35
     185 2235.07   199.5 2224.58   214.7 2215.12   227.5 2204.73   239.7 2197.27
   247.9 2190.67   251.9  2188.5   260.1 2186.61   288.6 2169.36   313.1 2148.55
   317.2 2147.14   333.5 2145.88   356.6 2135.02   366.1    2133   520.9 2133.03
   537.2    2134   541.3  2135.3   549.5  2139.1   565.8 2138.89   590.2 2143.29
   626.9 2142.64   781.8 2151.97   851.1 2159.91   880.4  2165.4     910 2172.76
#Mann= 8 ,-1,0
       0      .1       0     290    .025       0   356.6    .035       0
   541.3    .025       0     590      .1       0     610     .05       0
     690     .06       0     890      .1       0
Bank Sta=356.6,541.3
XS Rating Curve= 0 ,0
Exp/Cntr=0.3,0.1

Type RM Length L Ch R = 1 ,134094  ,496.2,497.1,498.2
XS GIS Cut Line= 2
     2239020.792      448074.794     2238885.413      448974.668
#Sta/Elev= 30
       0 2299.38    22.6 2280.25    42.9 2268.38      59 2260.39   111.7 2239.37
   144.9 2223.75   216.8 2192.82   227.7 2187.08   257.2 2168.72   265.3 2165.89
   285.6 2156.36   297.7 2148.71   305.8 2146.31   322.6 2146.35     326 2145.33
   338.1 2137.77   347.2 2134.76   361.3 2132.25   431.2 2132.19   547.6 2132.22
   556.6  2134.5   565.2 2138.28   576.8 2139.14   593.3 2143.94   621.5  2143.5
     771 2149.69   819.5 2155.55   839.7 2159.36     868 2161.29     910 2170.51
#Mann= 8 ,-1,0
       0      .1       0     270    .025       0   347.2    .035       0
   556.6      .1       0     570     .05       0     640      .1       0
     670     .05       0     870     .06       0
Bank Sta=347.2,556.6
XS Rating Curve= 0 ,0
Exp/Cntr=0.3,0.1

Type RM Length L Ch R = 1 ,133596  ,514.4,503.8,494.2
XS GIS Cut Line= 2
     2238533.678      447996.3062238372.62645478449011.122043254
#Sta/Elev= 30
       0 2272.92    37.3 2264.79   106.2 2243.68   150.7 2233.78   183.8 2223.94
   199.3  2217.2   215.3 2211.83   239.8  2198.7   260.1 2184.48   284.4 2162.18
   292.5 2155.61   304.6 2147.49   320.8 2145.29   337.6 2133.91     341 2132.15
   345.1 2131.62   539.5 2131.62  545.282133.831   554.3 2138.25   563.8 2138.08
     580 2143.41   588.1 2144.36   608.4 2143.51     657 2143.69   746.1 2146.28
   883.8 2144.47   956.7 2145.89   968.8 2148.75   994.8 2160.79  1027.5 2181.91
#Mann= 6 ,-1,0
       0      .1       0   337.6    .035       0  545.28    .025       0
     550     .05       0     850     .06       0     950      .1       0
Bank Sta=337.6,545.28
XS Rating Curve= 0 ,0
Exp/Cntr=0.3,0.1

Type RM Length L Ch R = 1 ,133093  ,516.1,499.6,482.2
XS GIS Cut Line= 2
     2237999.134      447922.1442237911.19018218449049.295473139
#Sta/Elev= 30
       0 2360.37    39.2 2339.58    83.3  2312.6   155.5  2264.8   191.6 2238.97
   219.7 2220.81   235.7 2206.22   243.8 2200.63   251.8 2192.86   267.8 2181.12
   275.9 2172.38   291.9  2151.1   295.9 2147.01     324 2142.65   340.5 2134.93
   344.1 2131.96     348 2131.07   548.7 2131.06   552.7 2131.19   560.1  2135.3
   568.8 2139.25   588.8  2144.3   905.8 2143.38  1010.1 2145.94  1022.1 2154.61
  1030.2  2162.8  1036.5 2167.63  1086.3 2203.04  1110.4 2218.95  1130.6 2230.44
#Mann= 7 ,-1,0
       0      .1       0     330    .025       0   340.5    .035       0
   560.1      .1       0     620     .05       0     920     .06       0
    1020      .1       0
Bank Sta=340.5,560.1
XS Rating Curve= 0 ,0
Exp/Cntr=0.3,0.1

Type RM Length L Ch R = 1 ,132593  ,499.6,469.8,437
XS GIS Cut Line= 3
     2237437.027      447902.5652237485.18292367448671.174630604
2237622.98452032449081.084654006
#Sta/Elev= 30
       0 2363.39    70.8 2323.87   110.8 2299.54   134.9  2278.1   166.9 2253.21
   235.1 2207.14   307.2 2154.74   315.2 2149.89   327.3 2144.99   351.3  2143.3
   359.3 2141.11   367.3 2133.27   371.3  2131.5   383.4 2130.16   539.7 2130.16
   555.7 2133.55   571.7 2136.56   583.8 2142.59   591.8 2144.09   683.5 2141.97
     756 2143.44   936.8 2142.23  1017.2 2143.89  1068.2 2142.04  1088.7 2142.34
  1102.5 2144.44  1122.5    2144  1126.7 2145.45  1168.9  2170.9  1202.6 2193.75
#Mann= 6 ,-1,0
       0      .1       0     340    .025       0   367.3    .035       0
   555.7      .1       0     740     .05       0 1050.12     .06       0
Bank Sta=367.3,555.7
XS Rating Curve= 0 ,0
Exp/Cntr=0.3,0.1

Type RM Length L Ch R = 1 ,132123  ,586.2,576.8,568.7
XS GIS Cut Line= 2
2236869.07108121448042.154362312 2237340.0501009449434.740476085
#Sta/Elev= 30
       0 2390.15    20.6 2369.86    72.1 2322.38   125.6 2277.51   163.7 2247.89
     197  2219.4   222.8 2194.71   246.9 2169.13     265 2162.87   282.5 2149.75
   310.9 2141.18   323.5  2131.4   332.6 2129.19   522.6 2129.22   526.8 2129.44
   528.6 2131.04   535.2 2139.18   543.7 2142.57   640.8 2140.45   695.7  2143.5
   813.9 2142.41   932.2 2143.47  1016.6 2145.97  1147.1 2152.87  1172.3 2155.81
  1185.5 2155.43  1276.5 2168.21  1317.5 2178.12  1371.3 2193.45  1470.1 2217.42
#Mann= 7 ,-1,0
       0      .1       0     320    .025       0   323.5    .035       0
   528.6      .1       0     590     .05       0    1150     .06       0
    1250      .1       0
Bank Sta=323.5,528.6
XS Rating Curve= 0 ,0
Exp/Cntr(USF)=0,0
Exp/Cntr=0.3,0.1

Type RM Length L Ch R = 1 ,131546  ,515.5,510.9,507.4
XS GIS Cut Line= 2
2236299.24461294448260.2002047612236828.36919062449481.256922474
#Sta/Elev= 30
       0 2407.09    53.4 2372.06    83.6  2347.7   129.2 2299.17   188.5 2243.74
   192.9  2238.4   197.2 2231.05   201.6 2226.63   253.8 2179.49   280.1 2158.64
   288.8 2144.65   293.1 2142.01   305.6 2140.56   318.32131.177     328  2128.5
   476.2 2128.51   488.1 2130.63   500.2 2133.04   525.5 2141.71   593.9 2138.81
   658.4 2143.58   942.7 2139.37  1029.9 2139.47  1064.8 2141.44  1077.8 2147.22
  1139.1 2182.05  1147.6 2184.86  1204.3 2186.12  1300.1 2182.79  1330.8 2184.54
#Mann= 7 ,-1,0
       0      .1       0     200    .025       0   318.3    .035       0
   488.1      .1       0     630     .05       0    1060     .06       0
    1160      .1       0
Bank Sta=318.3,488.1
XS Rating Curve= 0 ,0
Exp/Cntr(USF)=0,0
Exp/Cntr=0.3,0.1

Type RM Length L Ch R = 1 ,131036  ,434.1,440.8,448.1
XS GIS Cut Line= 2
2235755.58364577448344.5112638412236406.81389522449702.210042822
#Sta/Elev= 30
       0 2442.48    48.9 2434.14      85 2424.36   108.9 2414.25   132.9 2399.68
   243.8 2317.84   267.8 2297.46   311.3 2256.47   377.8 2199.16     400 2177.07
   404.4 2170.28   417.8 2144.96   422.2 2141.92   444.4 2140.75   460.6 2131.05
   473.1 2127.88   648.4 2127.88   660.92130.459   670.6 2134.52   692.8 2138.93
     806 2142.22   945.4  2140.5  1043.3  2137.3  1240.7 2141.42  1256.2 2145.32
    1274 2147.04  1341.1 2179.68  1371.6 2190.05  1433.7 2194.29  1505.8 2196.07
#Mann= 7 ,-1,0
       0      .1       0     330    .025       0   460.6    .035       0
   660.9      .1       0     760     .05       0    1200     .06       0
    1420     .05       0
#XS Ineff= 2 , 0
                         1221.51         2192.82
Permanent Ineff=
       F       F
Bank Sta=460.6,660.9
XS Rating Curve= 0 ,0
Exp/Cntr(USF)=0,0
Exp/Cntr=0.3,0.1

Type RM Length L Ch R = 1 ,130595  ,493.1,492.8,492.6
XS GIS Cut Line= 3
     2235417.329      448597.9262235709.64338889 449306.76402774
2236095.90094574449895.713864347
#Sta/Elev= 30
       0 2400.51    42.5 2370.51   111.7 2317.21   151.7 2290.09   194.6 2258.24
   219.1 2236.31   254.5 2207.23   271.2    2191   293.4 2172.12   297.7 2166.95
   310.7 2141.99   332.4 2139.95   338.6 2137.37   346.8 2131.22   350.8 2128.69
   358.3 2127.34     566 2127.34   570.3  2127.6   577.5 2131.49   587.6 2135.72
   609.3 2140.68   623.5  2141.2   848.3 2137.96   860.5  2136.5  1121.5 2144.03
  1166.1  2146.3  1296.1 2157.14  1319.2 2156.99  1458.5 2169.44  1471.1 2168.43
#Mann= 8 ,-1,0
       0      .1       0     260    .025       0   346.8    .035       0
   577.5    .025       0     580      .1       0     680     .05       0
 1256.75     .06       0 1376.75     .05       0
Bank Sta=346.8,577.5
XS Rating Curve= 0 ,0
Exp/Cntr=0.3,0.1

Type RM Length L Ch R = 1 ,130102  ,513.8,498.7,482.1
XS GIS Cut Line= 3
2234956.08222346 448774.788392942235383.45207466449803.964769298
2235685.80897619450245.871009994
#Sta/Elev= 30
       0 2399.36     106 2328.37   171.5 2280.48   193.2 2262.94   214.8 2244.57
   271.1    2189   289.6  2169.6     311  2143.1   314.4 2140.68   335.5 2138.85
     3522130.016   362.1 2126.72   561.3 2126.69   575.72129.542     583 2134.75
     596 2133.94   617.6 2141.17   623.1 2141.72   885.7 2137.94  1026.4 2138.76
    1300  2137.5  1328.2 2139.93    1363 2150.93  1382.4  2155.3  1491.1 2169.72
  1527.3 2177.26  1547.8 2177.48  1561.7 2180.29  1597.3 2182.58  1649.8 2181.05
#Mann= 9 ,-1,0
       0      .1       0     350    .025       0     352    .035       0
   575.7      .1       0     600     .06       0     610     .07       0
     710     .05       0 1494.38     .06       0 1644.38     .05       0
Bank Sta=352,575.7
XS Rating Curve= 0 ,0
Exp/Cntr(USF)=0,0
Exp/Cntr=0.3,0.1

Type RM Length L Ch R = 1 ,129603  ,524.8,508.7,491.9
XS GIS Cut Line= 2
     2234457.944      449021.1882235308.15172765450510.034832219
#Sta/Elev= 30
       0 2365.53    25.1 2351.18   136.5 2276.34   234.9 2194.23   278.8 2162.43
   294.8 2145.95   308.6 2140.28   344.7 2139.26359.59852129.144   373.1 2126.06
   529.7 2126.07562.91772128.442   571.2  2134.4     588 2139.59   598.8 2140.41
   806.1    2140  1004.2 2134.91  1068.9 2139.06  1253.6 2137.15  1312.8 2138.06
  1372.7 2135.99  1427.9 2137.33  1441.2 2139.45  1478.6 2161.34    1497 2169.66
  1515.4 2174.93  1537.1 2178.56  1593.8 2180.98  1685.9 2172.44  1714.5 2173.93
#Mann= 9 ,-1,0
       0      .1       0     240    .025       0359.5985    .035       0
562.9177      .1       0     580     .06       0     690     .05       0
    1470      .1       0    1490     .05       0    1710     .06       0
Bank Sta=359.5985,562.9177
XS Rating Curve= 0 ,0
Exp/Cntr=0.3,0.1

Type RM Length L Ch R = 1 ,129094  ,518.5,503.3,487.7
XS GIS Cut Line= 2
     2233976.226      449327.0682234979.08835519450629.375011813
#Sta/Elev= 30
       0 2420.93      10 2410.11    26.1 2395.99    58.5 2372.69    83.4 2351.39
   118.8  2324.8   176.9 2277.41   198.3 2257.43   229.4 2232.17     250 2212.63
   290.4  2177.2   309.5 2157.78   320.7 2142.81   340.9 2138.56   355.1  2129.7
   376.3 2125.59   524.4 2125.64     553 2129.06     558 2133.99   577.6 2138.97
   626.1 2140.01   862.8 2134.58   956.8 2138.75  1426.4 2134.97  1498.9 2136.08
  1507.4 2137.29  1521.7 2142.69  1560.2  2162.2  1581.6 2169.49  1643.7  2180.9
#Mann= 7 ,-1,0
       0      .1       0     250     .05       0   355.1    .035       0
     553     .06       0     700     .05       0    1490      .1       0
    1620     .05       0
Bank Sta=355.1,553
XS Rating Curve= 0 ,0
Exp/Cntr=0.3,0.1

Type RM Length L Ch R = 1 ,128591  ,518.2,502.6,490.2
XS GIS Cut Line= 2
     2233558.671      449701.1062234756.68178508450901.509125836
#Sta/Elev= 30
       0  2441.4      34 2397.58    57.7 2373.13    75.7 2357.75   119.9 2327.34
   158.3 2298.18   186.6 2278.94   209.2 2260.59     240 2239.64     294  2188.8
   310.9 2165.11   323.6 2141.72   329.2 2138.93   341.9 2137.33   354.7 2128.81
   370.2 2125.19   523.1 2125.24   535.7 2127.06   548.3 2126.01   559.6 2129.05
   578.1  2137.2   630.7 2139.66   729.1 2133.89   789.2 2138.56  1117.6 2136.87
  1177.7 2138.01  1469.4 2133.98    1548 2139.57    1585 2146.76  1695.9 2161.12
#Mann= 13 ,-1,0
       0      .1       0     310     .05       0   354.7    .035       0
   559.6     .06       0     640     .05       0     720     .06       0
     920     .05       0    1000      .1       0    1050     .05       0
    1140      .1       0    1190     .05       0    1420     .06       0
    1470      .1       0
Bank Sta=354.7,559.6
XS Rating Curve= 0 ,0
Exp/Cntr=0.3,0.1

Type RM Length L Ch R = 1 ,128089  ,344.5,337.5,335.2
XS GIS Cut Line= 4
2233328.55030448450164.2030556492233514.39854766450377.928535302
 2233663.0771422450484.7912751292234434.34735138451395.447666697
#Sta/Elev= 30
       0 2345.17    82.6  2281.7   105.3 2266.32   139.1  2240.1   150.7 2232.76
   170.5 2214.63   192.1 2190.78   218.7  2166.2   255.5 2139.24   273.7 2137.14
   286.8 2128.59   295.3  2124.9   301.2 2124.81   466.3 2124.81   473.1 2125.36
   478.7 2128.79   484.4 2130.88   507.1 2133.15   529.8    2138   595.1 2134.05
   660.4 2135.66  1001.5 2135.71  1230.8 2132.23  1398.3 2135.82  1415.3 2142.56
  1432.3 2145.68  1494.2 2167.98  1604.3 2189.39  1625.4  2190.2  1659.7 2199.58
#Mann= 11 ,-1,0
       0      .1       0  283.23     .05       0   286.8    .035       0
   478.7    .025       0  496.33      .1       0  626.33     .06       0
  756.33     .05       0 1276.33     .07       0 1306.33     .06       0
 1456.33      .1       0 1526.33     .06       0
Bank Sta=286.8,478.7
XS Rating Curve= 0 ,0
Exp/Cntr(USF)=0,0
Exp/Cntr=0.3,0.1

Type RM Length L Ch R = 1 ,127751  ,624.1,668.8,702
XS GIS Cut Line= 4
 2233189.1641221450494.083687288 2233323.9040984450661.347106148
 2233505.1061355450777.5022581332234109.11292582451576.649703795
#Sta/Elev= 30
       0 2267.66    29.7 2245.92   103.9 2185.42   138.7 2168.31     158 2155.77
   169.3 2146.63   189.7 2137.77   211.9  2136.9   229.3 2127.68   235.1 2125.17
   243.6 2124.53   435.1 2124.57   444.7 2128.02   449.7 2130.87   468.3 2135.78
   486.2 2136.59   554.5 2134.94  1065.9 2132.41  1181.7 2138.88  1205.9 2137.85
  1225.8 2143.71    1282 2150.16    1292 2153.31    1302 2158.72  1332.1 2168.36
  1348.6 2169.74  1377.2 2176.61  1403.7 2179.76  1417.4 2185.35  1431.7 2186.01
#Mann= 11 ,-1,0
       0      .1       0      50     .05       0     210    .025       0
   229.3    .035       0   444.7    .025       0  450.02     .06       0
  610.02     .05       0 1100.02     .06       0 1200.02      .1       0
 1330.02     .07       0 1430.02     .06       0
Bank Sta=229.3,444.7
XS Rating Curve= 0 ,0
Exp/Cntr(USF)=0,0
Exp/Cntr=0.3,0.1

Type RM Length L Ch R = 1 ,127082  ,459.1,487.6,510
XS GIS Cut Line= 2
     2232706.049      450868.7352233619.84510428 452045.72293357
#Sta/Elev= 30
       0 2191.72      23 2185.59    42.6 2175.53    55.6 2166.61    76.5 2159.15
     117 2138.49   167.7 2133.93   289.8 2134.19  319.12 2126.53   329.6 2124.09
   562.7 2124.12   567.7 2126.35   574.8 2131.48   593.1  2135.9   868.5 2134.82
     954 2130.61  1005.3 2130.72  1096.5 2134.67  1150.7 2145.91  1226.1 2145.68
  1236.2 2149.37    1259 2166.65  1266.6 2170.41    1302  2181.2  1321.7 2182.87
  1342.5 2192.58  1381.6 2194.02  1423.6 2218.24    1470 2235.11  1490.1 2244.96
#Mann= 10 ,-1,0
       0      .1       0  319.12    .035       0   567.7      .1       0
     670     .07       0     680     .06       0     790      .1       0
     920     .06       0    1160     .05       0    1290     .06       0
    1410      .1       0
Bank Sta=319.12,567.7
XS Rating Curve= 0 ,0
Exp/Cntr=0.3,0.1

Type RM Length L Ch R = 1 ,126595  ,471.5,506.3,534.3
XS GIS Cut Line= 2
 2232323.7562962451010.8688650042233011.11330881452321.667430106
#Sta/Elev= 30
       0  2176.7    25.2 2163.92    38.7 2142.82    43.3 2138.81    47.8  2137.5
    83.9 2136.95   115.5 2133.12   278.1 2134.97   363.9 2132.98   379.9 2131.33
   393.8 2126.36   405.7 2123.78   625.9 2123.88   634.9 2126.71   671.1  2134.9
   725.3 2132.53   779.5 2133.28   797.5 2129.78   811.1 2129.66   838.2 2130.97
   856.2 2135.45     915 2133.87   996.3 2135.22  1137.8 2141.63  1175.3  2144.9
  1287.9 2148.18  1344.6 2154.24  1398.2 2164.65  1456.5 2173.45  1480.1 2174.48
#Mann= 9 ,-1,0
       0      .1       0     210     .05       0   393.8    .035       0
   634.9    .025       0     660     .05       0     990     .06       0
    1080     .07       0    1100     .06       0    1210      .1       0
Bank Sta=393.8,634.9
XS Rating Curve= 0 ,0
Exp/Cntr=0.3,0.1

Type RM Length L Ch R = 1 ,126088  ,373.5,482.2,574.4
BEGIN DESCRIPTION:
channel burned 0.60' to transition from approximate to detailed reach:
lidar = 2123.47
interpolated = 2122.87
END DESCRIPTION:
XS GIS Cut Line= 3
2232031.93290826450958.2327549072232046.30848052451469.665259785
2232336.11109374452508.825851578
#Sta/Elev= 30
       0  2173.7      51 2168.57      59 2164.39      71 2147.29      75  2145.4
      87  2144.2      99 2136.78   143.2  2131.6   447.1  2133.7     542 2134.13
   552.7 2133.14   569.3 2127.55   581.7 2122.87   830.9 2122.96   840.7 2127.95
   847.5 2132.03   864.1 2135.82  1109.1 2132.76  1258.6 2133.07  1291.8 2136.42
    1325 2133.66  1352.4 2134.37  1370.7 2134.78  1420.6 2142.01  1466.2 2168.77
    1487 2184.62  1516.1 2185.78  1545.1 2210.12  1561.7 2219.56  1590.4 2235.81
#Mann= 8 ,-1,0
       0      .1       0   143.2     .05       0   447.1      .1       0
     542    .025       0   569.3    .035       0   840.7     .05       0
  1352.4     .06       0  1561.7      .1       0
Bank Sta=569.3,840.7
XS Rating Curve= 0 ,0
Exp/Cntr=0.3,0.1

Type RM Length L Ch R = 1 ,125606  ,268.2,339.7,408.7
BEGIN DESCRIPTION:
channel burned 1.21' to transition from approximate to detailed reach:
lidar = 2123.47
interpolated = 2122.01
END DESCRIPTION:
XS GIS Cut Line= 3
 2231801.0041363450932.7224600172231715.86523674451431.719624135
2231351.11936566452351.777994766
#Sta/Elev= 30
       0 2176.74    20.8 2174.32    45.1 2167.36    53.2 2162.35    70.4 2146.16
    84.3 2136.71   101.9 2135.51   114.1 2130.38   146.5 2132.81   170.9 2131.94
   223.6 2133.62   361.6 2131.84   576.6 2133.35   589.5 2133.88  599.91 2126.13
   606.7 2122.01   856.3 2122.07   864.9 2126.13   886.4 2129.55   946.7 2130.75
  1032.7 2128.04  1217.8 2130.47  1246.6 2128.88  1316.7 2130.81  1346.8  2132.1
  1359.7  2135.8  1381.3 2136.08  1385.6 2137.38  1417.1 2155.37  1495.9 2193.43
#Mann= 11 ,-1,0
       0     .05       0    70.4      .1       0   170.9     .05       0
   361.6      .1       0   576.6    .025       0  599.91    .035       0
   864.9      .1       0   886.4     .05       0  1246.6     .08       0
  1316.7     .06       0  1417.1      .1       0
Bank Sta=599.91,864.9
XS Rating Curve= 0 ,0
Exp/Cntr=0.3,0.1

Type RM Length L Ch R = 1 ,125266  ,394.9,405.3,413.8
BEGIN DESCRIPTION:
channel burned 1.63' to transition from approximate to detailed reach:
lidar = 2123.03
interpolated = 2121.40
END DESCRIPTION:
XS GIS Cut Line= 4
2231683.14945968450874.0700363652231522.16932687451299.009423998
2231009.21235665451773.211307584 2230232.7250924452081.005650681
#Sta/Elev= 30
       0 2161.87    37.5 2157.69    71.8 2155.96   114.5 2135.93   144.3 2130.99
     225 2132.25   240.5  2129.6     256 2132.12   401.1 2131.35   457.4 2130.75
   538.8  2131.5   547.9 2125.45   555.2  2121.4   822.1 2121.42     831 2126.01
   834.7 2128.27   853.6 2132.79  1204.8  2129.6  1230.8 2129.52  1317.6 2133.83
  1433.8 2134.12  1498.9 2132.71  1519.8 2138.21  1643.7 2139.61  1751.5 2136.54
  1795.2 2135.18    1821 2154.11  1885.6 2184.64  1971.6 2241.51  1988.2 2248.86
#Mann= 13 ,-1,0
       0     .06       0    37.5      .1       0   240.5     .05       0
   401.1      .1       0   457.4    .025       0   547.9    .035       0
     831      .1       0   834.7     .05       0  1204.8      .1       0
  1230.8     .05       0  1433.8      .1       0  1643.7     .08       0
  1751.5      .1       0
#XS Ineff= 2 , 0
                            1702         2152.15
Permanent Ineff=
       F       F
Bank Sta=547.9,831
XS Rating Curve= 0 ,0
Exp/Cntr=0.3,0.1

Type RM Length L Ch R = 1 ,124861  ,357,380.2,422.1
BEGIN DESCRIPTION:
channel burned 2.07' to transition from approximate to detailed reach:
lidar = 2122.75
interpolated = 2120.68
END DESCRIPTION:
XS GIS Cut Line= 3
2231479.12287281450838.2098702922230438.09034469451674.409609313
2230110.35788214451852.734625704
#Sta/Elev= 30
       0 2177.12      44 2174.15    49.5 2169.75    75.3 2140.19    81.4 2136.07
   112.3 2135.47   135.1 2128.16     266 2131.64   288.7 2128.38   297.3 2124.29
  306.42 2120.64   598.9 2120.71   605.2 2124.18   610.2 2131.67   615.9    2133
  1096.6 2129.12  1183.8 2131.95  1204.3 2133.58  1349.4 2135.93  1392.1 2132.69
  1427.2 2133.31  1446.8 2134.74  1460.4 2145.07  1537.8 2189.87  1592.5 2225.56
  1601.6 2229.12    1638 2256.09  1692.7 2288.48  1697.2 2292.64  1708.4 2308.62
#Mann= 7 ,-1,0
       0      .1       0   297.3    .035       0   605.2     .05       0
  1183.8     .03       0  1204.3     .08       0  1427.2     .06       0
  1537.8      .1       0
Bank Sta=297.3,605.2
XS Rating Curve= 0 ,0
Exp/Cntr(USF)=0,0
Exp/Cntr=0.3,0.1

Type RM Length L Ch R = 1 ,124481  ,493.9,497.3,513.4
BEGIN DESCRIPTION:
channel burned 1.93' to transition from approximate to detailed reach:
lidar = 2121.93
interpolated = 2120.0
END DESCRIPTION:
XS GIS Cut Line= 2
2231288.74886883450590.000725857 2229977.8190186451329.808564126
#Sta/Elev= 30
       0 2175.03      38 2174.12    51.2 2173.91   106.3 2167.37   114.3 2162.34
   140.7  2136.6   161.4 2134.74     189 2127.14   201.8 2129.49   208.3 2123.73
   211.9    2120   492.1 2120.19   501.3 2123.63   515.1  2132.2   628.1  2131.9
   636.2 2131.99   740.1 2131.93   830.7 2131.95   950.6 2131.65  1097.9 2130.11
  1125.9 2133.41  1191.9 2133.89  1235.9 2133.78  1291.7 2133.84  1364.8 2134.49
  1383.2 2150.22  1410.7 2163.35  1430.7 2172.24  1461.2 2185.92  1505.3  2214.1
#Mann= 16 ,-1,0
       0     .07       0      38     .06       0    51.2      .1       0
   161.4    .025       0   208.3    .035       0   501.3     .06       0
   628.1     .05       0   636.2     .08       0   740.1     .07       0
   830.7     .06       0   950.6     .05       0  1191.9      .1       0
  1235.9     .05       0  1291.7     .07       0  1410.7     .06       0
  1430.7      .1       0
Bank Sta=208.3,501.3
XS Rating Curve= 0 ,0
Exp/Cntr(USF)=0,0
Exp/Cntr=0.3,0.1

Type RM Length L Ch R = 1 ,123984  ,519.8,510.3,496.2
BEGIN DESCRIPTION:
channel burned 1.75' to transition from approximate to detailed reach:
lidar = 2120.86
interpolated = 2119.11
END DESCRIPTION:
XS GIS Cut Line= 2
2231228.88083474450069.6177563162229648.91719895450911.758855112
#Sta/Elev= 30
       0 2210.76    32.5  2203.9    64.3 2192.36      96 2190.61   210.1 2168.35
   263.3 2152.48     300 2150.39   322.6 2136.08   340.8 2134.83  357.71 2122.07
   363.4 2119.11     559 2119.13  570.28 2121.77   600.4 2121.57   653.5    2132
     726 2132.36     766 2132.38   875.4 2129.88     930 2129.36  1216.1 2131.58
  1321.9  2131.7  1351.4 2134.81  1543.6 2130.16  1560.1 2131.38  1590.9 2135.18
  1708.4 2230.75  1745.9 2264.42    1764 2276.97  1777.6 2298.16  1790.4 2308.43
#Mann= 15 ,-1,0
       0      .1       0      96     .06       0   322.6    .025       0
  357.71    .035       0  570.28    .025       0   653.5     .06       0
     726     .07       0     766     .06       0   875.4     .05       0
     930     .06       0  1216.1     .08       0  1321.9     .07       0
  1351.4     .08       0  1543.6     .07       0  1560.1      .1       0
#Block Obstruct= 1 ,-1
  741.59  754.41 2150.63
Bank Sta=357.71,570.28
XS Rating Curve= 0 ,0
Exp/Cntr=0.3,0.1

Type RM Length L Ch R = 1 ,123473  ,397.2,376.2,401.6
BEGIN DESCRIPTION:
start GRL detailed reach - channel burned 2.08':
lidar invert = 2120.28
effective invert = 2118.20
END DESCRIPTION:
XS GIS Cut Line= 3
2230836.33611434449672.6223597132230247.38332597450055.629840518
2229473.14840302450407.758978043
#Sta/Elev= 30
       0 2181.96    32.3 2170.19    62.2 2166.25    74.4 2156.68    90.1 2156.24
   105.2 2154.57   133.8 2136.07   162.4 2137.12     172 2134.45   181.5 2123.76
  189.33 2120.44   194.2 2118.22   377.1  2118.2  384.33 2120.46   428.4  2122.7
   448.7 2127.82   474.7 2127.11   584.5 2129.93   921.4 2127.73   965.3  2130.1
  1237.7 2130.47    1330 2131.27  1360.8 2132.44  1382.8    2133  1391.6 2138.24
  1406.9 2151.88  1435.5 2166.16  1453.1 2171.69  1488.9 2196.51  1553.1 2251.52
#Mann= 10 ,-1,0
       0      .1       0    74.4    .016       0    90.1      .1       0
  189.33    .035       0  384.33      .1       0   474.7     .05       0
  1237.7     .07       0    1330     .06       0  1360.8    .016       0
  1391.6      .1       0
#Block Obstruct= 1 ,-1
 1170.13 1244.98 2148.89
Bank Sta=189.33,384.33
XS Rating Curve= 0 ,0
Exp/Cntr(USF)=0,0
Exp/Cntr=0.3,0.1

Type RM Length L Ch R = 1 ,123097  ,708,580.1,320.7
BEGIN DESCRIPTION:
channel burned 2.29':
lidar invert = 2119.88
interpolated invert = 2117.59
END DESCRIPTION:
Node Name=T
XS GIS Cut Line= 3
     2230711.076      449232.9692230224.07711222  449654.0219267
2229342.18120445450024.676156277
#Sta/Elev= 30
       0 2194.91    72.6 2159.98    83.2 2152.75    93.7 2150.92   104.4 2150.08
   130.7 2141.14   141.3 2138.92   167.8 2134.99   210.1 2134.61   220.6 2134.66
   294.7    2131     300 2128.87  312.55 2119.99   315.8 2117.59   550.8 2117.59
  556.57 2120.04   569.6 2125.17   580.2 2127.42   611.9  2127.5   638.4 2130.86
   676.7 2128.64   777.5 2128.51  1134.9 2128.17  1171.6 2129.72  1455.1 2130.65
  1468.1 2130.14  1502.8 2151.36    1529 2170.93  1567.9 2203.83  1600.4 2235.05
#Mann= 11 ,-1,0
       0      .1       0    93.7    .016       0   104.4     .08       0
   141.3     .06       0   210.1    .016       0   220.6     .07       0
  312.55    .035       0  556.57      .1       0   611.9     .06       0
   777.5    .016       0  1455.1     .01       0
#XS Ineff= 2 , 0
          221.07  2145.9 1435.22         2148.83
Permanent Ineff=
       F       F
#Block Obstruct= 2 ,-1
  275.08  294.66 2149.56 1176.78 1298.36 2147.36
Bank Sta=312.55,556.57
XS Rating Curve= 0 ,0
Exp/Cntr=0.3,0.1

Type RM Length L Ch R = 1 ,122517  ,478.8,529.1,460.3
BEGIN DESCRIPTION:
channel burned 2.38':
lidar invert = 2119.03
interpolated invert = 2116.65
END DESCRIPTION:
XS GIS Cut Line= 4
2230551.67080971448426.8513351752230209.38546449448643.971145313
2229746.59856102449477.7221539492229270.25862493449824.632715939
#Sta/Elev= 30
       0 2235.01    15.8 2220.37    30.3 2218.01      42  2208.1    56.2 2205.43
    70.5 2193.24   114.4 2169.62     152 2148.58   168.6 2143.33   189.7 2142.73
   201.3 2142.27   226.8  2141.5   321.5 2129.87   383.1 2132.21   392.7 2132.25
   473.8 2129.47   507.4 2129.53   694.9 2129.67   717.8 2130.32   801.3  2130.1
   821.9 2121.46   836.8 2116.65  1070.1 2116.68  1080.8 2120.99  1120.4 2125.17
  1289.6 2127.25  1782.5 2128.48  1822.1 2129.08  1827.1 2131.33  1948.2 2233.81
#Mann= 15 ,-1,0
       0      .1       0   114.4     .08       0   189.7    .016       0
   201.3     .08       0   383.1    .016       0   392.7      .1       0
   473.8    .016       0   507.4     .06       0   694.9    .016       0
   717.8     .06       0   821.9    .035       0  1080.8     .08       0
  1120.4     .05       0  1289.6    .016       0  1827.1      .1       0
#XS Ineff= 2 , 0
          617.46 2142.39
Permanent Ineff=
       F       F
#Block Obstruct= 2 ,-1
  736.51   772.3 2147.67  1536.1 1577.96 2145.92
Bank Sta=821.9,1080.8
XS Rating Curve= 0 ,0
Exp/Cntr=0.3,0.1

Type RM Length L Ch R = 1 ,121988  ,298.1,470.5,574.8
BEGIN DESCRIPTION:
channel burned 2.04':
lidar invert = 2117.84
effective invert = 2115.80
END DESCRIPTION:
XS GIS Cut Line= 5
2230360.64513631448074.2694426242229596.68277897448599.372905041
2229464.89517095448885.5994126882229265.14579271449334.498237478
2229026.27587978449447.750621024
#Sta/Elev= 30
       0 2213.05    49.1 2190.48   146.2 2158.13   157.8 2148.98   165.6 2147.03
   183.7 2146.35   214.1 2127.74   304.5 2127.26   354.9 2131.28   393.6 2127.38
   524.8 2129.45   563.6 2129.13   727.3    2130   845.1  2132.1   968.6  2131.5
  1028.3 2129.64  1065.5 2119.97  1100.8 2119.87  1105.2 2115.93    1465  2115.8
  1478.1 2118.39    1535 2118.45  1665.8 2126.88  1739.7 2128.76  1756.7 2129.16
  1796.3 2132.27  1823.1 2158.85  1840.8 2169.98  1969.2 2282.45  1997.8 2312.84
#Mann= 15 ,-1,0
       0      .1       0   165.6    .016       0   183.7      .1       0
   304.5     .08       0   524.8    .016       0   563.6     .05       0
   727.3     .07       0   845.1     .05       0   968.6      .1       0
  1100.8    .035       0  1478.1     .08       0  1665.8    .016       0
  1739.7     .05       0  1756.7    .016       0  1796.3      .1       0
#Block Obstruct= 3 ,-1
  470.72  523.36 2148.09  604.99  807.19 2149.53 1544.04 1566.32 2139.48
Bank Sta=1100.8,1478.1
XS Rating Curve= 0 ,0
Exp/Cntr(USF)=0,0
Exp/Cntr=0.3,0.1

Type RM Length L Ch R = 1 ,121517  ,485.6,488.3,492.1
BEGIN DESCRIPTION:
channel burned 1.12':
lidar invert = 2116.04
interpolated invert = 2114.92
END DESCRIPTION:
XS GIS Cut Line= 2
2230284.62765637447685.9612300112228712.42605681448974.379849421
#Sta/Elev= 30
       0  2283.8     8.3  2281.2    52.3 2245.51   144.7 2182.11   181.8 2160.01
   204.4 2141.62   269.5 2137.22   289.7  2136.2     338  2135.2   367.8 2126.25
   448.9 2130.53   465.8 2130.43   525.6 2128.82   957.3 2129.34  1196.4 2131.71
  1292.5 2129.74  1311.4 2122.59  1329.7 2118.13  1349.9 2122.13  1486.3 2118.17
  1503.3 2114.94  1696.6 2114.92    1709 2117.97    1725 2129.92  1734.2 2132.22
  1765.8 2132.72  1787.6  2151.6  1835.2 2184.12  1992.9 2316.91  2032.7 2345.16
#Mann= 12 ,-1,0
       0      .1       0   269.5    .016       0   289.7      .1       0
   448.9    .016       0   465.8     .07       0   525.6    .016       0
   957.3     .05       0  1311.4      .1       0  1486.3    .035       0
    1709     .06       0  1734.2    .016       0  1765.8      .1       0
#Block Obstruct= 2 ,-1
  234.76  237.07 2157.94  586.34  688.25 2147.86
Bank Sta=1486.3,1709
XS Rating Curve= 0 ,0
Exp/Cntr=0.3,0.1

Type RM Length L Ch R = 1 ,121029  ,440,467.3,469.2
BEGIN DESCRIPTION:
channel burned 1.61':
lidar invert = 2115.61
effective invert = 2114.0
END DESCRIPTION:
Node Name=S
XS GIS Cut Line= 2
2229961.13089064447328.8140883862228476.45907868448541.725936561
#Sta/Elev= 30
       0 2191.79    57.8  2147.9    94.2 2137.21   101.7 2137.12   117.5 2135.68
   140.2 2126.05   254.3 2126.69     271  2129.2   285.2 2128.91   373.3  2126.5
   404.1 2126.92   533.2  2126.7   546.7  2126.4   670.8 2126.99   739.8  2127.3
  1333.8 2125.48  1364.8 2131.02  1380.3 2120.29  1393.9 2118.13    1432    2114
  1602.4 2117.03  1617.9 2129.73  1631.8 2132.79  1661.1 2132.59  1690.2 2148.69
  1716.1 2151.32  1732.2 2159.96  1764.5 2186.92  1871.5 2256.89  1917.1 2291.57
#Mann= 16 ,-1,0
       0      .1       0    94.2    .016       0   101.7      .1       0
   254.3     .08       0     271    .016       0   285.2     .05       0
   373.3    .016       0   404.1     .05       0   533.2    .016       0
   546.7     .05       0   670.8    .016       0   739.8     .05       0
  1393.9    .035       0  1602.4     .07       0  1631.8    .016       0
  1661.1      .1       0
#Block Obstruct= 3 ,-1
  301.34   354.3 2146.74  418.04  465.71 2145.18  617.64  674.92 2145.98
Bank Sta=1393.9,1602.4
XS Rating Curve= 0 ,0
Exp/Cntr(USF)=0,0
Exp/Cntr=0.3,0.1

Type RM Length L Ch R = 1 ,120562  ,378.3,379,373.7
BEGIN DESCRIPTION:
channel burned 1.89':
lidar invert = 2115.17
interpolated invert = 2113.28
END DESCRIPTION:
XS GIS Cut Line= 2
2229806.70213926446917.6708005822228139.20012199448206.862888825
#Sta/Elev= 30
       0 2220.06   143.1 2131.62   195.4  2126.9   260.8 2127.65   336.9 2127.97
   341.9 2127.85   352.3 2127.06   372.1 2130.46   468.4 2130.58   494.8 2125.65
   548.5  2125.1   672.8 2125.26   691.5 2125.37     817 2126.53   865.5 2127.13
   993.8 2127.71   999.5 2127.72  1150.9 2123.91  1176.3 2124.03  1176.3 2124.02
  1432.9 2125.07  1455.7 2117.04  1472.8 2113.28  1647.2 2113.32  1655.3 2117.01
  1686.7 2132.22  1723.7 2133.09  1732.4 2137.53  1752.6 2152.32  2107.7 2341.74
#Mann= 19 ,-1,0
       0      .1       0   195.4    .016       0   260.8     .05       0
   336.9    .016       0   341.9     .05       0   352.3    .016       0
   548.5     .06       0   672.8    .016       0   691.5     .06       0
     817    .016       0   865.5     .06       0   993.8    .016       0
   999.5     .06       0  1150.9    .016       0  1176.3     .06       0
  1455.7    .035       0  1655.3     .06       0  1686.7    .016       0
  1732.4      .1       0
#Block Obstruct= 7 ,-1
  263.73  308.34 2145.72  378.38   492.3 2148.58  570.65  677.87 2143.49
  759.01  815.02 2145.39  875.72  938.72 2145.26 1010.02 1053.07 2146.38
 1220.43 1380.85 2142.92
Bank Sta=1455.7,1655.3
XS Rating Curve= 0 ,0
Exp/Cntr(USF)=0,0
Exp/Cntr=0.3,0.1

Type RM Length L Ch R = 1 ,120183  ,403,389.9,380.3
BEGIN DESCRIPTION:
structure xs 4 - channel burned 2.14':
lidar invert = 2114.84
effective invert = 2112.70
END DESCRIPTION:
XS GIS Cut Line= 4
2229568.08121917 446617.160021412228580.41036262 447395.28035205
2228208.14290035447681.2140299492227995.75631452447858.523945553
#Sta/Elev= 30
       0 2223.33    71.2 2172.58   106.8 2142.63   122.8 2133.16   157.7 2127.12
   187.9 2125.69   202.2  2125.5   310.3 2127.09     356 2123.88   417.4 2125.87
   686.4 2125.14  1001.9 2127.11  1186.4  2123.7  1333.3 2125.05  1375.8 2121.69
  1390.1 2118.09  1404.4 2112.71  1621.2  2112.7  1626.9 2112.88  1635.9 2117.92
  1646.8 2121.66  1656.1  2127.4  1667.6 2128.74  1698.2 2129.14  1726.8 2130.69
  1747.6 2135.84  1789.3 2156.26  1826.6  2177.6  1920.2 2233.89  2003.4 2288.04
#Mann= 11 ,-1,0
       0      .1       0   122.8     .08       0   187.9    .016       0
   202.2     .06       0   310.3    .016       0  1186.4     .06       0
  1390.1    .035       0  1635.9     .08       0  1667.6    .016       0
  1698.2     .07       0  1747.6      .1       0
#XS Ineff= 2 , 0
          253.87 2143.41 1670.42         2142.71
Permanent Ineff=
       F       F
#Block Obstruct= 7 ,-1
  388.22  462.22 2143.54  584.54  657.87 2143.13  769.83  818.99 2143.44
  891.42  950.86 2144.57  983.92 1003.96 2144.96 1056.66 1088.11 2143.78
 1702.88 1726.77 2148.55
Bank Sta=1390.1,1635.9
XS Rating Curve= 0 ,0
Exp/Cntr(USF)=0,0
Exp/Cntr=0.5,0.3

Type RM Length L Ch R = 1 ,119793  ,120.9,107.3,102.7
BEGIN DESCRIPTION:
structure xs 3
END DESCRIPTION:
XS GIS Cut Line= 3
2229640.08411498446315.3449802252229258.10127402446337.382451819
2227671.40331926447630.247451994
#Sta/Elev= 30
       0 2388.21   144.1 2305.66   282.8  2219.6   340.5 2183.67   389.5 2138.29
   409.4 2136.76   439.3 2126.87   470.9 2126.42    1190  2125.5  1453.2 2127.73
  1515.1 2128.41 1568.24  2123.4 1576.55 2120.11 1587.16 2115.51  1609.6 2113.23
 1722.55 2110.68 1845.21 2112.23 1864.11 2120.11 1902.73 2127.28  1978.1 2127.74
  2092.6 2131.56  2108.5 2132.17    2121 2137.27  2129.5 2135.16  2196.2 2171.65
  2269.3 2226.88  2288.3  2235.2  2311.5 2239.42  2379.7 2282.93  2429.3 2306.53
#Mann= 11 ,-1,0
       0      .1       0   282.8     .06       0   470.9    .016       0
    1190     .05       0  1453.2    .016       0  1515.1     .05       0
 1576.55    .035       0 1864.11     .08       0 1902.73      .1       0
  1978.1    .016       0  2092.6      .1       0
#XS Ineff= 2 , 0
          1512.2 2124.63  1930.8          2128.6
Permanent Ineff=
       F       F
#Block Obstruct= 7 ,-1
  431.67  500.53 2149.33  707.36  751.35 2145.42  794.28  823.42 2144.86
  887.17 1003.34  2144.5 1028.88 1132.46 2145.41 1204.91 1261.48 2147.23
 2091.67  2132.8 2157.17
Bank Sta=1576.55,1864.11
XS Rating Curve= 0 ,0
Exp/Cntr(USF)=0,0
Exp/Cntr=0.5,0.3

Type RM Length L Ch R = 3 ,119745  ,,,
BEGIN DESCRIPTION:
Bridge No.: 54075GRL050 8th Street
JV notes: road deck updated per surveyed XS data points
channel burned per surveyed cross sections
structure opening based on survey data, photos, and aerial imagery
surveyed inverts are 3-4' below inverts from lidar:
 surveyed invert US is 2110.71
 surveyed invert DS is 2111.04
END DESCRIPTION:
Bridge Culvert--1,0,-1,-1, 0
Deck Dist Width WeirC Skew NumUp NumDn MinLoCord MaxHiCord MaxSubmerge Is_Ogee
28,40,2.6,0, 435, 435, , , 0.98, 0, 0,0,,
   -12.4    -7.3    -3.3      .7     4.7    10.9    16.7    20.7    24.7    28.7
    32.7    36.7    40.7    44.7    52.7    56.7    60.7    64.7    68.7    72.7
    76.7    80.7    84.7    88.7    96.7   100.7   102.7   106.7   110.7   112.7
   114.7   118.8   120.7   122.8   124.7   128.7   130.8   136.7   140.7   144.7
   148.7   152.7   156.7   160.7   164.7   168.7   172.7   176.7   180.7   182.8
   184.7   188.7   192.7   194.7   198.8   200.7   204.7   206.7   210.8   212.7
   220.7   224.7   228.7   232.7   236.7   240.7   244.7   248.7   252.7   258.6
   264.7   268.7   270.9   272.7   284.7   286.6   288.7   290.9   294.6   298.6
   304.7   308.7   312.7   316.7   320.7   324.7   328.7   336.7   340.7   344.7
   346.5   348.7   352.7     355   356.7     359   363.7   364.8     369     371
   373.8   376.2   377.7     379   382.4   384.2   386.2   389.1   391.9     395
   397.6   399.8   403.3   407.5   411.8   413.8   417.5   420.1   430.9   441.3
   445.1   451.4   454.4   457.3   460.1   465.8   472.5   477.7   482.9   491.3
     497   498.4   503.6   508.8   514.1   522.6   528.3   534.8     540   545.5
   548.2   556.7   562.4   565.2   571.2   576.8   581.5   585.1   587.9   597.1
   602.3   607.5   612.7   616.3   628.3   636.2   644.8   649.1   659.5   669.8
     675   684.5   687.4   695.9   706.2   711.4   716.6   718.6     727   732.8
   737.4   739.9   744.2   752.9   763.3   772.6   775.4   778.9   785.7   792.5
   799.7   809.5   815.1   821.4   825.7   829.4   830.9   833.9     836   837.9
   843.6   851.6   857.8   860.7   866.3   872.4   877.8   882.8     888   889.1
   891.9   896.7   898.4   906.1   911.8   915.5   923.2     928   934.3   946.8
   950.3   960.7   965.9   971.9   976.3   982.8   994.2  1008.4  1012.6  1025.4
  1028.3  1033.4  1039.6  1048.2  1053.8  1059.7  1065.2  1073.7  1084.8  1087.9
  1093.6  1096.5  1100.9    1105  1113.5  1128.7  1137.3  1141.9  1144.7  1147.7
  1150.4  1153.8  1158.1  1163.3  1172.6  1181.7  1189.2  1197.7  1207.2  1210.2
  1212.9  1216.5  1221.5  1222.7  1227.1  1230.8  1235.7  1241.5  1249.9  1255.5
  1260.4  1266.6  1272.9    1284  1291.7    1298    1301  1310.5  1315.2  1329.5
  1335.6  1346.5  1360.7    1372  1376.2  1381.4  1386.6  1398.3  1404.6  1414.6
  1423.4  1428.1  1443.7  1448.5  1454.1  1464.5  1469.7  1475.2 1518.62 1541.19
 1541.19 1621.14 1637.68 1721.45  1737.5 1770.23 1821.66 1837.23 1901.63 1917.98
 1941.63 1941.63 1957.44 2007.84  2008.4  2014.1  2022.6  2030.6  2036.8  2044.2
  2051.4  2056.7    2063  2065.2    2068  2072.2  2073.7  2079.4  2085.1  2087.8
  2093.6  2096.4  2102.1  2107.8  2110.6  2116.3  2118.9  2125.7  2130.5  2133.4
  2134.5  2136.2  2141.9  2144.6  2147.6  2150.8  2156.1  2160.5  2163.4  2164.6
  2167.5  2169.6  2173.1  2176.1  2178.8  2181.7  2184.5  2186.4  2187.4  2191.6
  2194.7  2195.9  2196.8  2198.7    2201    2202  2204.4  2207.3  2210.1  2212.4
  2215.8  2217.6  2218.6  2222.8  2224.3  2227.1    2230  2232.3  2235.6  2238.6
  2241.3  2243.6  2248.8  2252.7    2254  2259.2  2261.2  2264.1  2266.9    2270
  2272.6  2276.2  2278.3  2283.9  2285.1  2286.8  2288.8  2289.6  2295.5  2298.1
  2300.7  2301.3  2307.6  2309.5  2312.4  2313.9  2316.3  2320.1  2321.5  2323.7
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                                                                         2128.13
 2128.13 2128.11 2128.11 2128.09 2128.09 2128.09 2128.08 2128.07 2128.06
    29.6    34.7    38.7    42.7    46.7    52.9    58.7    62.7    66.7    70.7
    74.7    78.7    82.7    86.7    94.7    98.7   102.7   106.7   110.7   114.7
   118.7   122.7   126.7   130.7   138.7   142.7   144.7   148.7   152.7   154.7
   156.7   160.8   162.7   164.8   166.7   170.7   172.8   178.7   182.7   186.7
   190.7   194.7   198.7   202.7   206.7   210.7   214.7   218.7   222.7   224.8
   226.7   230.7   234.7   236.7   240.8   242.7   246.7   248.7   252.8   254.7
   262.7   266.7   270.7   274.7   278.7   282.7   286.7   290.7   294.7   300.6
   306.7   310.7   312.9   314.7   326.7   328.6   330.7   332.9   336.6   340.6
   346.7   350.7   354.7   358.7   362.7   366.7   370.7   378.7   382.7   386.7
   388.5   390.7   394.7     397   398.7     401   405.7   406.8     411     413
   415.8   418.2   419.7     421   424.4   426.2   428.2   431.1   433.9     437
   439.6   441.8   445.3   449.5   453.8   455.8   459.5   462.1   472.9   483.3
   487.1   493.4   496.4   499.3   502.1   507.8   514.5   519.7   524.9   533.3
     539   540.4   545.6   550.8   556.1   564.6   570.3   576.8     582   587.5
   590.2   598.7   604.4   607.2   613.2   618.8   623.5   627.1   629.9   639.1
   644.3   649.5   654.7   658.3   670.3   678.2   686.8   691.1   701.5   711.8
     717   726.5   729.4   737.9   748.2   753.4   758.6   760.6     769   774.8
   779.4   781.9   786.2   794.9   805.3   814.6   817.4   820.9   827.7   834.5
   841.7   851.5   857.1   863.4   867.7   871.4   872.9   875.9     878   879.9
   885.6   893.6   899.8   902.7   908.3   914.4   919.8   924.8     930   931.1
   933.9   938.7   940.4   948.1   953.8   957.5   965.2     970   976.3   988.8
   992.3  1002.7  1007.9  1013.9  1018.3  1024.8  1036.2  1050.4  1054.6  1067.4
  1070.3  1075.4  1081.6  1090.2  1095.8  1101.7  1107.2  1115.7  1126.8  1129.9
  1135.6  1138.5  1142.9    1147  1155.5  1170.7  1179.3  1183.9  1186.7  1189.7
  1192.4  1195.8  1200.1  1205.3  1214.6  1223.7  1231.2  1239.7  1249.2  1252.2
  1254.9  1258.5  1263.5  1264.7  1269.1  1272.8  1277.7  1283.5  1291.9  1297.5
  1302.4  1308.6  1314.9    1326  1333.7    1340    1343  1352.5  1357.2  1371.5
  1377.6  1388.5  1402.7    1414  1418.2  1423.4  1428.6  1440.3  1446.6  1456.6
  1465.4  1470.1  1485.7  1490.5  1496.1  1506.5  1511.7  1517.2 1560.62 1583.19
 1583.19 1663.14 1679.68 1763.45  1779.5 1812.23 1863.66 1879.23 1943.63 1959.98
 1983.63 1983.63 1999.44 2049.84  2050.4  2056.1  2064.6  2072.6  2078.8  2086.2
  2093.4  2098.7    2105  2107.2    2110  2114.2  2115.7  2121.4  2127.1  2129.8
  2135.6  2138.4  2144.1  2149.8  2152.6  2158.3  2160.9  2167.7  2172.5  2175.4
  2176.5  2178.2  2183.9  2186.6  2189.6  2192.8  2198.1  2202.5  2205.4  2206.6
  2209.5  2211.6  2215.1  2218.1  2220.8  2223.7  2226.5  2228.4  2229.4  2233.6
  2236.7  2237.9  2238.8  2240.7    2243    2244  2246.4  2249.3  2252.1  2254.4
  2257.8  2259.6  2260.6  2264.8  2266.3  2269.1    2272  2274.3  2277.6  2280.6
  2283.3  2285.6  2290.8  2294.7    2296  2301.2  2303.2  2306.1  2308.9    2312
  2314.6  2318.2  2320.3  2325.9  2327.1  2328.8  2330.8  2331.6  2337.5  2340.1
  2342.7  2343.3  2349.6  2351.5  2354.4  2355.9  2358.3  2362.1  2363.5  2365.7
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                                                                         2128.13
 2128.13 2128.11 2128.11 2128.09 2128.09 2128.09 2128.08 2128.07 2128.06
Pier Skew, UpSta & Num, DnSta & Num=  ,1633.54, 2 ,1697.39, 2 , 0 , 0 , 0 ,,
     2.5     2.5
       0  2128.5
     2.5     2.5
       0  2128.5
Pier Skew, UpSta & Num, DnSta & Num=  ,1733.85, 2 ,1797.7, 2 , 0 , 0 , 0 ,,
     2.5     2.5
       0  2128.5
     2.5     2.5
       0  2128.5
Pier Skew, UpSta & Num, DnSta & Num=  ,1843.06, 2 ,1897.91, 2 , 0 , 0 , 0 ,,
     2.5     2.5
       0  2128.5
     2.5     2.5
       0  2128.5
BR Coef=-1 ,-1 , 0 ,, 0 ,,,0.8,0,1.33,0,
WSPro=,,,, 1 ,,,, 0 ,,,, 0 ,,,,-1 ,-1 ,-1 , 0 , 0 , 0 , 0 , 0
BC Design=,, 0 ,, 0 ,,,,,,
BC Use User HTab Curves=0
BC User HTab FreeFlow(D)= 0

Type RM Length L Ch R = 1 ,119686  ,429.9,441.7,444.3
BEGIN DESCRIPTION:
structure xs 2
END DESCRIPTION:
XS GIS Cut Line= 3
2229607.02790759446216.1763580522229228.71797857446190.465974526
2227642.02002381447531.078829821
#Sta/Elev= 30
       0    2329    95.1    2301   239.4  2240.4   287.5 2216.86   332.1 2188.71
   355.7 2162.86   367.7 2157.96   379.9 2137.45   395.6 2130.21     427 2126.29
   569.3 2122.65   678.4 2125.37   720.3 2125.62  1343.7 2127.24  1449.4 2122.73
  1589.5 2127.05 1638.42 2121.94 1704.59 2112.37 1803.26 2111.04 1908.15 2112.38
 1945.32 2121.61  1962.52126.352  2155.5 2131.31  2217.9 2160.38  2249.4 2168.32
  2271.9 2184.64  2304.7 2194.77  2354.3 2223.71  2390.7 2237.46  2456.4 2283.24
#Mann= 11 ,-1,0
       0      .1       0   239.4     .08       0   332.1      .1       0
     427    .016       0   678.4     .05       0   720.3    .016       0
  1589.5     .08       0 1638.42    .035       0 1945.32     .08       0
  1962.5    .016       0  2155.5      .1       0
#XS Ineff= 2 , 0
          1570.8 2124.45    1956          2127.8
Permanent Ineff=
       F       F
#Block Obstruct= 9 ,-1
  449.85  576.09 2145.52  791.04   889.5  2145.8  998.36 1071.46 2144.92
 1108.74 1210.62 2145.07 1291.85 1401.34 2146.73 1410.84 1452.61 2145.67
 1483.13  1532.6 2145.26 1580.08 1639.42 2147.56 1970.49 2087.43 2149.15
Bank Sta=1638.42,1945.32
XS Rating Curve= 0 ,0
Exp/Cntr(USF)=0,0
Exp/Cntr=0.5,0.3

Type RM Length L Ch R = 1 ,119244  ,687.6,730,720.6
BEGIN DESCRIPTION:
xs 1 - channel burned = 2.78':
lidar invert = 2113.58
effective invert = 2110.80
END DESCRIPTION:
XS GIS Cut Line= 3
2229725.89807675446172.0696783222228734.21185503 446058.20940842
2227283.41164176447240.887050626
#Sta/Elev= 30
       0 2319.74   203.4 2265.06     356 2208.93   376.2 2200.32     452    2132
   476.8 2123.84     964 2125.05   988.2 2123.85  1010.3 2127.52  1027.3 2124.84
  1034.6 2123.19  1354.3 2121.31  1568.5 2124.38    1704 2122.04  1717.7 2121.69
  1979.8 2121.46 1995.052115.798    2002  2110.8  2262.7 2110.92  2270.4 2115.52
  2306.5 2122.01  2477.3 2124.97  2522.3  2126.8  2531.3    2132  2556.9 2132.75
  2565.4 2133.63  2641.9 2174.69  2719.3 2227.08  2753.1 2242.61    2870  2335.9
#Mann= 17 ,-1,0
       0      .1       0     356     .08       0     452      .1       0
   476.8    .016       0     964     .05       0  1010.3    .016       0
  1027.3     .05       0  1034.6    .016       0  1568.5     .06       0
    1704    .016       0  1717.7      .1       0 1995.05    .035       0
  2270.4      .1       0  2306.5     .07       0  2477.3     .06       0
  2531.3    .016       0  2556.9      .1       0
#Block Obstruct= 6 ,-1
  753.43  824.42 2141.05 1282.92 1316.89 2139.51 1330.97 1387.82 2140.29
 1605.29 1637.91 2142.17 2420.88 2449.49 2142.43 2467.83 2511.33 2143.29
Bank Sta=1995.05,2270.4
XS Rating Curve= 0 ,0
Exp/Cntr(USF)=0,0
Exp/Cntr=0.3,0.1

Type RM Length L Ch R = 1 ,118514  ,364.1,357.5,357.4
BEGIN DESCRIPTION:
channel burned 2.72':
lidar invert =  2112.12
effective invert = 2109.4
END DESCRIPTION:
XS GIS Cut Line= 3
2229777.31884381446113.3030874052228205.31253678 445613.78706461
2226758.18523544446715.660644305
#Sta/Elev= 30
       0 2287.08   244.6 2195.29   287.7 2174.98   306.8 2148.99   325.9 2134.14
   367.3 2124.72     572 2131.06     614 2123.29     807 2125.22  1109.4 2123.92
  1220.9 2121.74  1331.7 2115.89    1403 2128.25  1440.8 2118.78  1524.7 2118.96
  1554.1 2119.26  1902.3 2123.25  1909.6 2123.22  2052.3 2124.46  2108.4 2125.44
  2216.3 2124.59  2240.7 2124.47  2415.1 2115.36  2425.1  2109.4 2659.752115.246
  3048.3 2125.83  3229.5 2139.49  3279.4 2141.82    3305 2141.64  3468.3 2190.03
#Mann= 19 ,-1,0
       0      .1       0   367.3    .016       0     572     .05       0
     614    .016       0     807     .05       0  1109.4    .016       0
  1220.9      .1       0  1524.7    .016       0  1554.1     .05       0
  1902.3    .016       0  1909.6     .06       0  2052.3    .016       0
  2108.4     .06       0  2216.3    .016       0  2240.7     .06       0
  2415.1    .035       0 2659.75      .1       0  3229.5    .016       0
  3279.4      .1       0
#XS Ineff= 2 , 0
           565.2 2138.01
Permanent Ineff=
       F       F
#Block Obstruct= 10 ,-1
   617.3  729.54  2141.8   812.9 1109.55 2143.67  1575.4 1582.13 2136.88
 1664.42 1704.88 2138.26 1877.74  1905.1 2140.55 1918.35 1941.68 2140.49
 1979.26 2037.69 2141.93 2116.57 2176.09 2142.35 2253.42  2276.5 2141.57
 2919.44  2981.2 2140.78
Bank Sta=2415.1,2659.75
XS Rating Curve= 0 ,0
Exp/Cntr(USF)=0,0
Exp/Cntr=0.3,0.1
