HEC-RAS study GRNBRRRV.prj: GRNBRRRV

--- GRNBRRRV.g01 (geometry) --- (continued)

Type RM Length L Ch R = 1 ,84090   ,353.1,406.8,423.6
BEGIN DESCRIPTION:
channel burned 4.57':
lidar invert = 2070.22
interpolated invert = 2065.65
END DESCRIPTION:
XS GIS Cut Line= 3
2216387.96353418423596.2891984172216010.95685021423945.214036957
     2215939.539      424614.576
#Sta/Elev= 30
       0 2210.86    70.6 2178.67   172.1 2127.48     193 2113.49   212.3 2089.11
   217.7 2088.13   228.6 2086.88   255.9 2071.24   326.7 2071.41   348.6 2076.19
   362.8 2073.79     390 2078.79   448.9 2079.64     570 2076.64   622.3 2078.61
   666.5 2072.12   674.6 2065.83   683.4 2065.65   847.5 2065.79   852.8 2072.36
   859.6 2075.99   903.9 2078.86     928 2085.12   992.4 2084.91  1061.4 2088.52
  1073.4 2089.95  1094.1 2092.35  1121.1  2095.4  1165.3 2107.38  1186.9 2108.13
#Mann= 11 ,-1,0
       0      .1       0   217.7    .016       0   228.6      .1       0
   255.9     .04       0   326.7      .1       0   666.5    .035       0
   852.8      .1       0   903.9     .06       0  1061.4    .016       0
  1073.4     .06       0  1094.1      .1       0
#Block Obstruct= 1 ,-1
  967.64 1011.33 2101.01
Bank Sta=666.5,852.8
XS Rating Curve= 0 ,0
Exp/Cntr=0.3,0.1

Type RM Length L Ch R = 1 ,83683   ,212.7,479,559.6
BEGIN DESCRIPTION:
channel burned 3.09':
lidar invert = 2069.69
effective invert = 2066.6
END DESCRIPTION:
XS GIS Cut Line= 3
2216202.49160581423301.7244633362215643.00850394423802.403034978
2215510.27827857424501.336879955
#Sta/Elev= 30
       0 2230.68    56.8 2206.32   207.1 2124.06   215.1 2118.26   239.2 2093.81
   255.4 2087.48   264.7 2086.99   271.5 2084.99   282.2 2076.53   295.9 2070.06
   366.7 2070.12   373.5 2072.94   425.1 2079.92   486.2 2078.01   511.2 2081.69
   904.3 2083.43   928.7 2082.64   957.2 2074.33   981.9 2071.61   993.8  2066.6
  1152.6 2066.66  1156.7 2071.98  1168.9  2079.2  1193.6 2081.87    1230  2092.8
  1246.3 2092.23  1327.7 2126.71  1356.2 2141.76  1385.2 2161.84  1462.2 2223.25
#Mann= 9 ,-1,0
       0      .1       0   255.4    .016       0   264.7      .1       0
   295.9     .04       0   366.7      .1       0   981.9    .035       0
  1156.7      .1       0    1230    .016       0  1246.3      .1       0
Bank Sta=981.9,1156.7
XS Rating Curve= 0 ,0
Exp/Cntr(USF)=0,0
Exp/Cntr=0.3,0.1

Type RM Length L Ch R = 1 ,83204   ,224.3,379.5,402.4
BEGIN DESCRIPTION:
channel burned 2.66':
lidar invert = 2069.03
interpolated invert = 2066.37
END DESCRIPTION:
Node Name=G
XS GIS Cut Line= 2
  2216068.081251423197.5564383642214960.87595331423998.978178878
#Sta/Elev= 30
       0 2211.13    64.1 2172.19   137.2 2122.22   162.9 2097.07   176.7 2087.89
   182.6  2087.2   197.3    2087   228.8 2071.29   236.9 2069.31   326.2 2071.18
   334.8 2075.81   370.2 2080.76   725.8 2083.72   873.9 2081.51     931    2071
   938.1 2066.37  1056.7 2066.37  1065.3 2071.03  1076.7 2075.77  1099.6  2100.9
  1125.7  2124.7    1134 2128.76  1150.4  2129.1  1209.7 2191.23    1259 2233.67
  1268.9 2243.85  1281.9 2261.79  1298.5 2278.61    1343 2320.18  1366.8 2336.94
#Mann= 9 ,-1,0
       0      .1       0   182.6    .016       0   197.3      .1       0
   228.8     .04       0   326.2      .1       0     931    .035       0
  1065.3      .1       0    1134    .016       0  1150.4      .1       0
Bank Sta=931,1065.3
XS Rating Curve= 0 ,0
Exp/Cntr(USF)=0,0
Exp/Cntr=0.3,0.1

Type RM Length L Ch R = 1 ,82824   ,279.9,221,223.4
BEGIN DESCRIPTION:
channel burned 2.70':
lidaar invert = 2068.47
interpolated invert = 2065.77
END DESCRIPTION:
XS GIS Cut Line= 3
2215980.71452038423022.822977119 2215540.5206084423296.684075031
2214809.66430416423533.582325372
#Sta/Elev= 30
       0 2250.84   165.5 2122.94   185.1 2099.23   198.5 2088.27   203.2  2087.5
   217.3 2086.86     249 2069.92   336.1 2069.66   350.6 2076.79   373.8 2079.66
   531.4 2082.22   758.5 2078.02   817.3  2080.4   868.4 2070.88   880.4 2065.88
  1006.6 2065.77    1015 2070.65    1024 2073.31  1038.9 2088.33  1065.3 2105.59
  1090.7 2126.75  1103.4 2127.13  1107.5 2128.83  1124.3 2147.15  1160.6 2174.13
  1196.3 2208.66  1225.2 2229.78  1233.6 2244.71  1250.4 2262.16  1286.7 2282.27
#Mann= 9 ,-1,0
       0      .1       0   203.2    .016       0   217.3      .1       0
     249     .04       0   336.1      .1       0   868.4    .035       0
    1015      .1       0  1090.7    .016       0  1103.4      .1       0
Bank Sta=868.4,1015
XS Rating Curve= 0 ,0
Exp/Cntr(USF)=0,0
Exp/Cntr=0.3,0.1

Type RM Length L Ch R = 1 ,82603   ,350.8,237.4,206.7
BEGIN DESCRIPTION:
channel burned 4.96':
lidar invert = 2068.28
interpolated invert = 2063.32
END DESCRIPTION:
XS GIS Cut Line= 3
2215710.31292051422804.7147371732215337.22494676423137.071778702
2214819.17001446423292.515281864
#Sta/Elev= 30
       0 2190.59    21.7 2176.35    84.9 2127.38   115.4 2091.68   120.7 2087.34
     133 2086.82     139 2085.51   166.2 2069.88   249.3 2069.83     254 2072.27
   265.4 2072.38   286.8 2080.52   313.4 2081.31   426.8 2078.03   504.9 2079.74
   630.2 2077.22     672 2069.89   680.5 2063.41   781.5 2063.32   826.5 2063.35
   835.2 2070.12   843.2 2074.08   889.7 2121.79   898.9 2128.81   912.7 2130.08
   918.4    2131   947.1 2161.77   985.2 2194.46  1002.2 2211.91  1040.5 2243.61
#Mann= 9 ,-1,0
       0      .1       0   120.7    .016       0     133      .1       0
   166.2     .04       0   249.3      .1       0     672    .035       0
   835.2      .1       0   898.9    .016       0   912.7      .1       0
Bank Sta=672,835.2
XS Rating Curve= 0 ,0
Exp/Cntr=0.3,0.1

Type RM Length L Ch R = 1 ,82366   ,294,278.8,278.1
BEGIN DESCRIPTION:
channel burned 7.30':
lidar invert = 2068
effective invert = 2060.7
END DESCRIPTION:
XS GIS Cut Line= 3
2215760.61756439422522.1444054772215382.58844151422624.632301014
2214745.81938563423217.717991584
#Sta/Elev= 30
       0 2150.25    71.3 2153.55   137.2 2145.18   182.2 2148.83   249.1 2143.85
   286.4 2132.17   315.4 2127.72   344.4 2104.45   385.9 2085.03   407.9 2085.57
   427.7 2079.41     473  2079.6   504.3 2074.87   609.6 2076.74   826.8 2070.08
   826.8 2070.06   832.1 2060.96   838.1  2060.7   979.9  2060.8   982.5 2061.06
   988.1 2069.92  1010.8  2085.5  1050.4 2124.87  1058.9 2127.79  1064.5 2134.46
  1089.2 2179.28  1104.2 2190.32  1116.5 2205.22  1182.1 2229.33  1261.9 2232.74
#Mann= 7 ,-1,0
       0      .1       0   385.9    .016       0   407.9      .1       0
   826.8    .035       0   988.1      .1       0  1050.4    .016       0
  1058.9      .1       0
#XS Ineff= 2 , 0
          407.23 2107.85
Permanent Ineff=
       F       F
Bank Sta=826.8,988.1
XS Rating Curve= 0 ,0
Exp/Cntr(USF)=0,0
Exp/Cntr=0.3,0.1

Type RM Length L Ch R = 1 ,82087   ,530.7,482.2,464.9
BEGIN DESCRIPTION:
channel burned 5.09':
lidar invert = 2067.79
interpolated invert = 2062.70
END DESCRIPTION:
XS GIS Cut Line= 3
2215161.50690605422166.0147016932215033.12151902422564.147641353
     2214487.561      423092.627
#Sta/Elev= 30
       0 2114.53    82.5 2086.15   108.4  2079.9   158.8 2078.36   179.8 2082.44
   196.7 2078.19   221.9 2077.47   241.9 2084.79   264.2 2084.44   284.9 2075.39
   385.8 2073.28   428.2  2075.5     663 2068.61     667 2068.18   671.5  2062.7
   803.9 2062.84   807.3 2069.05   826.2  2080.4     861 2109.57   872.3 2109.87
   876.3  2112.2   891.2 2131.05   903.4 2159.58   906.3 2163.37   962.8 2199.66
   994.7 2214.12  1022.3 2212.84  1048.9 2204.66  1121.2 2191.88  1177.9 2196.56
#Mann= 7 ,-1,0
       0      .1       0   241.9    .016       0   264.2      .1       0
     663    .035       0   807.3      .1       0     861    .016       0
   872.3      .1       0
#XS Ineff= 2 , 0
          256.11 2096.39
Permanent Ineff=
       F       F
Bank Sta=663,807.3
XS Rating Curve= 0 ,0
Exp/Cntr=0.3,0.1

Type RM Length L Ch R = 1 ,81605   ,524.7,511.6,507.3
BEGIN DESCRIPTION:
channel burned 3.12':
lidar invert = 2067.44
interpolated invert = 2064.32
END DESCRIPTION:
XS GIS Cut Line= 2
     2214701.609      422105.5492214220.32104797422780.853987514
#Sta/Elev= 30
       0 2116.21      38 2090.84    48.7 2085.29    52.4 2084.82    64.5 2084.47
    97.8 2078.24   181.3 2074.16   205.8 2077.32   235.3 2075.73   253.1 2072.63
   289.3 2074.64   318.8 2069.12   323.7 2064.49   327.7 2064.32   551.4 2064.37
   554.6 2064.48     560 2069.45   581.4 2073.66   595.2 2078.43   608.6 2079.04
   614.5 2080.02   633.2 2091.76   691.7 2134.56   698.6 2140.54   706.9 2153.12
   743.6 2180.69   753.7 2191.61     810 2227.29   822.6 2239.43   829.3 2243.57
#Mann= 7 ,-1,0
       0      .1       0    52.4    .016       0    64.5      .1       0
   318.8    .035       0     560      .1       0   595.2    .016       0
   608.6      .1       0
Bank Sta=318.8,560
XS Rating Curve= 0 ,0
Exp/Cntr=0.3,0.1

Type RM Length L Ch R = 1 ,81094   ,405.4,501,583.5
BEGIN DESCRIPTION:
channel burned 2.61':
lidar invert = 2067.06
interpolated invert = 2064.45
END DESCRIPTION:
XS GIS Cut Line= 3
     2214256.745      421813.199     2214009.927      422195.437
      2213763.11      422577.676
#Sta/Elev= 30
       0 2143.48    14.3 2131.11    61.9 2099.06    75.6 2086.91    84.3  2084.1
     100 2083.77   104.6 2083.04   114.3 2078.81   123.8 2077.06   192.8 2078.03
   228.5 2076.95   280.9  2078.7   295.5 2076.92   314.2 2068.37   320.6 2064.58
   323.8 2064.45     579 2064.46   581.9 2064.69   585.6  2068.5   599.9 2073.29
   616.7 2074.03   642.6 2075.61   654.3 2075.78   694.8 2078.47   731.1 2084.95
   745.8 2086.27   780.9 2095.11   842.7 2119.97   890.4 2134.29     910 2141.77
#Mann= 9 ,-1,0
       0      .1       0    84.3    .016       0     100      .1       0
   314.2    .035       0   585.6     .07       0   616.7     .06       0
   642.6    .016       0   654.3     .06       0   731.1      .1       0
Bank Sta=314.2,585.6
XS Rating Curve= 0 ,0
Exp/Cntr=0.3,0.1

Type RM Length L Ch R = 1 ,80593   ,479.3,489.9,518.2
BEGIN DESCRIPTION:
channel burned 1.46':
lidar invert = 2065.69
interpolated invert = 2064.23
END DESCRIPTION:
XS GIS Cut Line= 3
     2213997.025      421610.3972213440.74808315422012.391857839
2213264.75146774422286.030903189
#Sta/Elev= 30
       0 2177.03    42.7 2146.85      57 2133.11    74.2 2126.73    91.4 2111.88
   125.8 2091.88   134.5 2085.06   140.1 2083.39   157.3 2083.54   171.6 2078.93
   191.7 2076.64   346.4 2077.28   352.1  2076.1   366.4 2068.05   372.2 2064.51
   603.1 2064.23     613 2064.28   619.4 2068.03   635.7 2072.02   687.4 2073.59
   739.6 2072.61   776.1 2066.07   853.7 2066.01   872.7 2070.73   894.4 2089.05
   901.3  2091.3   910.2 2091.36     916 2091.19   929.8 2103.73  1011.7 2156.81
#Mann= 9 ,-1,0
       0      .1       0   140.1    .016       0   157.3      .1       0
   366.4    .035       0   619.4      .1       0   776.1     .04       0
   853.7      .1       0   901.3    .016       0   910.2      .1       0
Bank Sta=366.4,619.4
XS Rating Curve= 0 ,0
Exp/Cntr=0.3,0.1

Type RM Length L Ch R = 1 ,80103   ,534.3,528.9,572
BEGIN DESCRIPTION:
channel burned 2.05':
lidar invert = 2064.78
interpolated invert = 2062.73
END DESCRIPTION:
XS GIS Cut Line= 4
     2213807.594      421220.4322213111.52471375421605.564172303
2213030.14856582421776.2550617162212645.91093217422046.755010801
#Sta/Elev= 30
       0 2262.25   123.7 2183.82   218.8 2139.28   232.5 2136.94   291.9 2108.04
   323.9  2084.6   332.7 2082.87   346.8 2082.78   355.9  2079.6   374.2 2066.64
   378.8 2062.82   457.1 2062.73   502.2 2062.79512.78252066.704   666.8 2071.39
   680.5  2069.3   799.5 2068.22   815.7 2065.29   919.2 2065.07   932.5 2074.36
  1041.8 2075.82  1055.6 2075.53  1084.9    2066  1207.2 2066.26    1268 2092.65
  1280.5 2092.72  1326.7 2106.27  1359.9 2109.44    1380 2122.81  1454.5 2155.79
#Mann= 11 ,-1,0
       0      .1       0   332.7    .016       0   346.8      .1       0
   374.2    .035       0512.7825      .1       0   815.7     .04       0
   919.2      .1       0  1084.9     .04       0  1207.2      .1       0
    1268    .016       0  1280.5      .1       0
Bank Sta=374.2,512.7825
XS Rating Curve= 0 ,0
Exp/Cntr=0.3,0.1

Type RM Length L Ch R = 1 ,79574   ,394.5,380.1,275.6
BEGIN DESCRIPTION:
channel burned 3.08':
lidar invert = 2064.04
interpolated invert = 2060.96
END DESCRIPTION:
Node Name=F
XS GIS Cut Line= 4
     2213520.183      420748.1642212840.42270359421172.985534124
 2212589.0309682421195.7710590212212065.72251591421748.440091361
#Sta/Elev= 30
       0 2273.55   203.9 2146.07   218.5 2141.86   259.4 2120.35   320.8 2097.15
   339.6 2082.32   349.1 2081.47   363.2 2081.45389.1935 2064.95   392.6 2060.96
   514.2 2060.98517.89142064.953   537.7 2070.62   583.1 2068.74   613.3 2071.31
     783 2069.87     813 2066.16    1049 2065.55  1064.1 2074.71  1163.1 2072.51
    1436 2074.56  1562.1 2080.39  1624.3 2090.94  1635.7 2095.26  1654.5 2108.14
    1664 2109.07  1678.4 2119.86  1700.5 2122.72  1717.7 2139.15  1815.1 2202.27
#Mann= 9 ,-1,0
       0      .1       0   349.1    .016       0   363.2      .1       0
389.1935    .035       0517.8914      .1       0     813     .04       0
    1049      .1       0  1654.5    .016       0    1664      .1       0
Bank Sta=389.1935,517.8914
XS Rating Curve= 0 ,0
Exp/Cntr=0.3,0.1

Type RM Length L Ch R = 1 ,79194   ,549.7,547.1,545.7
BEGIN DESCRIPTION:
channel burned 1.46':
lidar invert = 2063.26
effective invert = 2061.80
END DESCRIPTION:
XS GIS Cut Line= 2
2213247.84433321420409.0090760042211841.51376906421560.208874087
#Sta/Elev= 30
       0 2239.75    88.7 2184.27     134 2147.64   144.9 2145.17     165 2132.79
   206.3 2113.97     250 2097.95   275.6 2081.72   294.2 2080.97   320.1 2064.58
   325.2  2061.8   428.4  2061.8   521.3  2061.8   578.5 2062.15   588.9 2065.16
   614.7 2070.84     676 2068.64   694.9 2064.77     827 2064.56   920.8 2072.21
  1048.9 2071.13  1328.1 2078.95  1489.3 2077.09  1534.8 2079.19  1605.9 2089.84
  1648.5 2110.25  1671.3 2126.16  1682.6 2126.74  1705.4 2146.53  1817.4 2226.33
#Mann= 11 ,-1,0
       0      .1       0   275.6    .016       0   294.2      .1       0
   320.1    .035       0   428.4     .08       0   521.3    .035       0
   588.9      .1       0   694.9     .04       0     827      .1       0
  1671.3    .016       0  1682.6      .1       0
#XS Ineff= 2 , 0
                         1474.65         2125.15
Permanent Ineff=
       F       F
Bank Sta=320.1,588.9
XS Rating Curve= 0 ,0
Exp/Cntr(USF)=0,0
Exp/Cntr=0.3,0.1

Type RM Length L Ch R = 1 ,78647   ,444.3,439.1,424.7
BEGIN DESCRIPTION:
channel burned 1.46':
lidar invert = 2061.76
effective invert = 2060.3
END DESCRIPTION:
XS GIS Cut Line= 2
2212951.35349194 419949.019379022211537.47818567 421111.13464498
#Sta/Elev= 30
       0 2245.19    42.2 2227.19    76.6 2204.35   118.9 2182.06   154.3 2155.65
     175 2150.61   255.3 2081.89   272.4 2079.55   278.5 2077.94   297.9    2064
   308.9  2060.3   511.5 2060.51  520.062064.142     531 2067.73   630.2 2072.32
   656.5 2064.66   698.6 2063.63   801.5 2062.16     817 2065.27   822.2 2066.85
   832.6 2077.45   880.5 2076.82  1511.4 2077.78  1640.3 2078.93  1670.6 2084.05
  1724.6 2108.84  1780.1  2141.3  1811.2 2164.19  1820.8 2164.67  1830.2 2171.85
#Mann= 11 ,-1,0
       0      .1       0   255.3    .016       0   272.4    .045       0
   297.9    .035       0  520.06      .1       0   698.6     .04       0
     817      .1       0   880.5     .06       0  1511.4     .08       0
  1811.2    .016       0  1820.8      .1       0
#XS Ineff= 2 , 0
                          1480.8         2111.89
Permanent Ineff=
       F       F
Bank Sta=297.9,520.06
XS Rating Curve= 0 ,0
Exp/Cntr=0.3,0.1

Type RM Length L Ch R = 1 ,78207   ,460.8,470.1,505.5
BEGIN DESCRIPTION:
channel burned 0.06':
lidar invert = 2060.16
effective invert = 2060.1
END DESCRIPTION:
XS GIS Cut Line= 3
2212596.53489789419653.9879471712212044.78868836420151.804076072
 2211530.3786885420465.013390505
#Sta/Elev= 30
       0 2166.33    28.6  2160.8      49 2152.26    67.7 2150.43    84.6  2140.6
   145.9 2121.01     154 2116.34   186.6 2082.65   192.3 2079.62   205.2 2078.87
   212.1 2076.45   232.1 2061.97   242.9  2060.1     383 2060.13   392.9 2062.04
   404.7 2061.91   420.7 2066.99   428.7 2062.15   436.9 2060.22   515.1 2060.32
   523.1 2061.94   542.2 2062.71   560.1 2069.68   582.3 2067.82   603.9 2075.29
  1010.8 2074.62  1193.4 2077.88  1226.2 2081.74  1305.8 2102.46  1345.4 2104.55
#Mann= 7 ,-1,0
       0      .1       0   192.3    .016       0   205.2      .1       0
   232.1    .035       0   392.9      .1       0   428.7     .04       0
   523.1     .06       0
#Block Obstruct= 1 ,-1
  1340.3 1345.39 2124.49
Bank Sta=232.1,392.9
XS Rating Curve= 0 ,0
Exp/Cntr(USF)=0,0
Exp/Cntr=0.3,0.1

Type RM Length L Ch R = 1 ,77737   ,414.5,408.1,425
BEGIN DESCRIPTION:
channel burned 0.62':
lidar invert = 2059.62
effective invert = 2059.0
END DESCRIPTION:
XS GIS Cut Line= 2
2212285.39981733419334.5559311262211437.03816433419987.939600308
#Sta/Elev= 30
       0 2176.11    37.1 2158.11      52 2143.95    56.9 2138.83    62.1 2136.84
    82.6 2136.58   122.3 2114.21   151.1 2087.82   159.6 2081.37   165.3  2079.6
   179.6  2079.2   187.9 2076.48   199.5 2066.49   210.82061.086   218.6    2059
   417.3 2059.04   430.6  2061.1   440.8 2062.97   456.2 2065.96   470.5 2073.72
   476.1 2074.47   561.5 2072.19     668 2073.81   698.3 2069.73     791 2074.48
   902.4 2079.53   920.4 2086.02   955.4  2090.2  1040.1 2094.34  1070.8  2094.9
#Mann= 11 ,-1,0
       0      .1       0      52     .12       0   122.3    .025       0
   165.3    .016       0   179.6      .1       0   210.8    .035       0
   430.6      .1       0   440.8     .05       0     791     .06       0
   920.4     .05       0  1040.1     .06       0
#Block Obstruct= 2 ,-1
  830.42  859.96  2097.7  878.34  903.35 2099.03
Bank Sta=210.8,430.6
XS Rating Curve= 0 ,0
Exp/Cntr(USF)=0,0
Exp/Cntr=0.3,0.1

Type RM Length L Ch R = 1 ,77329   ,326,324.9,344.9
BEGIN DESCRIPTION:
channel burned 1.73':
lidar invert = 2059.16
interpolated invert = 2057.43
END DESCRIPTION:
XS GIS Cut Line= 2
2212129.83227705418967.4165360612211098.93804345419676.804519745
#Sta/Elev= 30
       0 2092.07    16.6 2085.14    62.9 2077.02    84.6 2076.48    99.1 2079.01
   118.5 2078.94   128.3 2076.45   212.4 2076.74   229.7 2073.62   235.4 2068.74
   239.9  2066.3   252.7  2063.9   259.4 2060.78   264.2 2057.46   269.1 2057.43
   511.2 2057.46   521.6 2060.73   531.3 2064.54     541 2071.69   551.8 2073.46
   642.9 2072.19   767.6 2072.22   880.9 2075.14   951.6 2078.51   982.8 2079.47
  1003.4 2081.64  1060.9 2084.71  1167.3 2095.31  1202.7 2096.26  1251.4 2099.88
#Mann= 7 ,-1,0
       0      .1       0    99.1    .016       0   118.5     .07       0
   212.4      .1       0   259.4    .035       0   521.6     .05       0
   951.6     .08       0
#XS Ineff= 2 , 0
          110.84 2082.44
Permanent Ineff=
       F       F
Bank Sta=259.4,521.6
XS Rating Curve= 0 ,0
Exp/Cntr(USF)=0,0
Exp/Cntr=0.3,0.1

Type RM Length L Ch R = 1 ,77004   ,366.1,413.5,435.6
BEGIN DESCRIPTION:
channel burned 1.99':
lidar invert = 2058.78
interpolated invert = 2056.79
END DESCRIPTION:
XS GIS Cut Line= 2
2212165.92918546418613.5952903662210931.00124203419315.133564484
#Sta/Elev= 30
       0 2124.93    11.2 2122.91    20.4 2115.11    29.6 2109.74    43.4 2106.08
    75.6 2084.54    89.4 2078.08   135.4 2071.86     163 2079.04   181.4 2078.66
   190.6 2075.51   203.4 2074.71   250.4 2076.44   296.4 2074.19     309 2075.55
   412.2 2075.23   435.2 2065.31   453.1 2060.42   458.6 2056.98   462.1 2056.82
   696.7 2056.79   705.1 2060.73   733.5 2071.84   903.7 2070.59   981.9 2072.45
  1073.9 2071.87    1198 2078.53  1259.6 2089.07  1359.1 2101.34  1420.3 2111.74
#Mann= 7 ,-1,0
       0      .1       0     163    .016       0   181.4     .07       0
   412.2      .1       0   453.1    .035       0   705.1     .05       0
    1198      .1       0
#XS Ineff= 2 , 0
          159.72 2086.88
Permanent Ineff=
       F       F
#Block Obstruct= 1 ,-1
  337.93  377.25 2093.17
Bank Sta=453.1,705.1
XS Rating Curve= 0 ,0
Exp/Cntr=0.3,0.1

Type RM Length L Ch R = 1 ,76591   ,157.7,521.5,638.5
BEGIN DESCRIPTION:
channel burned 2.05':
lidar invert = 2058
interpolated invert = 2055.95
END DESCRIPTION:
XS GIS Cut Line= 3
2212383.18025794418408.5650161132211833.21683358418376.259882991
2210797.58636298418825.496629003
#Sta/Elev= 30
       0 2117.02   123.2 2119.08   275.5 2116.26   295.5 2104.55   308.8 2106.54
   315.5 2104.85   343.6 2082.33   351.6 2079.98   363.6 2080.48   371.6 2079.65
   391.7 2071.99   415.7 2072.84   730.8 2074.32   770.1 2073.19   792.6 2063.07
   813.7 2060.37   831.1 2055.95  1040.4 2056.04  1051.7 2061.21  1066.3 2068.21
  1105.9 2069.63  1230.5 2069.65  1333.9  2066.7  1445.9 2070.49  1476.9 2079.64
  1507.3 2095.13  1525.5 2111.51  1576.7 2146.19  1594.1 2163.63  1679.8 2219.91
#Mann= 9 ,-1,0
       0      .1       0   351.6    .016       0   363.6      .1       0
   415.7     .05       0   730.8      .1       0   813.7    .035       0
  1051.7      .1       0  1105.9     .05       0  1445.9      .1       0
Bank Sta=813.7,1051.7
XS Rating Curve= 0 ,0
Exp/Cntr=0.3,0.1

Type RM Length L Ch R = 1 ,76069   ,234.3,471.8,524.9
BEGIN DESCRIPTION:
channel burned 3.57':
lidar invert = 2057
interpolated invert = 2053.43
END DESCRIPTION:
Node Name=E
XS GIS Cut Line= 2
2212399.14354824418380.1229354142210944.50363709417887.550024203
#Sta/Elev= 30
       0  2114.9    45.4 2111.78   277.6  2107.1   294.5 2099.97   310.7 2100.19
   339.1 2081.75   345.2 2079.68   367.5 2079.69   383.2 2072.38     417 2071.49
   754.8 2075.57   875.4 2070.39     928 2070.27   936.4 2068.76   953.3 2060.24
   982.9 2061.65   994.4 2059.09    1011 2053.52  1194.1 2053.43  1200.3 2053.75
  1210.9 2059.04  1232.1 2068.43    1249 2078.81  1312.3 2134.53  1316.5 2139.47
    1325 2155.12  1332.8 2164.31  1455.9 2285.69  1502.3 2314.61  1535.8 2318.92
#Mann= 7 ,-1,0
       0      .1       0   345.2    .016       0   367.5      .1       0
     417     .05       0     928      .1       0   994.4    .035       0
  1210.9      .1       0
Bank Sta=994.4,1210.9
XS Rating Curve= 0 ,0
Exp/Cntr=0.3,0.1

Type RM Length L Ch R = 1 ,75598   ,488.5,612.5,635.7
BEGIN DESCRIPTION:
channel burned 3.46':
lidar invert = 2056.17
interpolated invert = 2052.71
END DESCRIPTION:
XS GIS Cut Line= 2
2212289.25609668418288.7794192672211425.38241124417459.099499966
#Sta/Elev= 30
       0 2105.94   140.1 2099.11   150.4 2095.75   164.6 2095.29   201.3 2079.72
     207 2079.32   228.9 2079.51   245.5 2072.31   276.6 2071.64   605.9 2074.43
   713.4 2073.59   758.7 2069.64   816.8 2067.86   832.2 2060.86   857.7 2059.85
   872.2 2057.17   877.2 2052.77  1001.9 2052.71  1021.8  2052.8  1024.6 2057.06
  1041.6 2061.86  1050.4 2066.64  1069.8 2093.63  1092.5 2118.44  1112.3 2144.96
  1137.7 2165.18  1151.9 2187.13    1183 2214.31    1189 2217.58  1197.8 2225.33
#Mann= 7 ,-1,0
       0      .1       0     207    .016       0   228.9      .1       0
   276.6     .05       0   758.7      .1       0   872.2    .035       0
  1024.6      .1       0
Bank Sta=872.2,1024.6
XS Rating Curve= 0 ,0
Exp/Cntr=0.3,0.1

Type RM Length L Ch R = 1 ,74985   ,425.5,438.1,446.4
BEGIN DESCRIPTION:
channel burned 3.41':
lidar invert = 2055.28
interpolated invert = 2051.87
END DESCRIPTION:
XS GIS Cut Line= 3
 2212553.6902218418070.4786928692212495.32781171417926.927204466
2212004.03370752417116.012700592
#Sta/Elev= 30
       0 2094.99      85 2089.69   175.7 2086.98   185.1 2083.47   203.8 2080.61
   234.3 2080.22   245.9  2084.1   254.6 2084.19   361.8 2073.23   560.4 2069.79
   616.5 2071.37   708.9 2069.38   732.2 2070.41   746.3 2068.36     765 2059.74
   778.9 2058.82   786.3 2062.97   793.4  2064.1813.79822056.971   821.1 2051.98
   928.7 2051.87   984.8 2051.89  988.65 2052.48993.39822056.895  1003.5 2060.18
  1017.9 2069.39  1025.6 2078.59  1045.6 2107.52  1092.4 2160.74  1103.1 2170.58
#Mann= 7 ,-1,0
       0      .1       0   203.8    .016       0   234.3      .1       0
   361.8     .05       0   732.2      .1       0813.7982    .035       0
993.3982      .1       0
#XS Ineff= 2 , 0
          254.38 2090.99
Permanent Ineff=
       F       F
Bank Sta=813.7982,993.3982
XS Rating Curve= 0 ,0
Exp/Cntr(USF)=0,0
Exp/Cntr=0.3,0.1

Type RM Length L Ch R = 1 ,74547   ,227.5,281.9,305.1
BEGIN DESCRIPTION:
channel burned 3.77':
lidar invert = 2054.97
effective invert = 2051.20
END DESCRIPTION:
XS GIS Cut Line= 3
2212862.35987121417887.3959238152212840.89535518417747.956639902
2212396.06390903 416893.86225307
#Sta/Elev= 30
       0 2090.02    62.9 2083.93   143.7 2084.64   157.7 2081.66   184.8 2080.14
     206 2080.34   225.4 2077.95   261.5  2078.3   315.8 2073.33   401.7 2070.48
   659.7 2069.72   712.5 2069.94     726 2065.59   753.1 2062.61   766.1 2063.58
   784.6 2062.24   807.2 2057.03   816.2 2051.31   960.5  2051.2   988.8 2051.28
   996.6 2056.77  1005.6 2060.97  1017.2 2071.98  1023.7 2079.39  1043.2 2106.86
  1059.7 2126.56  1073.3 2140.28  1091.3 2155.48  1103.8 2161.62  1104.1 2161.66
#Mann= 8 ,-1,0
       0      .1       0   184.8    .016       0     206      .1       0
   261.5     .07       0   659.7      .1       0   807.2    .035       0
   996.6      .1       0  1103.8      .1       0
#XS Ineff= 2 , 0
          255.55 2085.83
Permanent Ineff=
       F       F
Bank Sta=807.2,996.6
XS Rating Curve= 0 ,0
Exp/Cntr(USF)=0,0
Exp/Cntr=0.3,0.1

Type RM Length L Ch R = 1 ,74265   ,215.8,230.5,246.4
BEGIN DESCRIPTION:
xs 4 - channel burned 3.88':
lidar invert = 2054.73
interpolated invert = 2050.85
END DESCRIPTION:
XS GIS Cut Line= 4
2212872.90673913417873.3088946382212872.90673913417783.878814313
2212920.25207577417601.5115916892212694.04657847416780.859089879
#Sta/Elev= 30
       0 2087.78    56.1  2084.7   141.8 2085.47   207.9 2082.29   228.6  2078.6
   286.5 2079.87   307.4 2076.88   358.4 2076.83   460.3 2072.94   502.2 2070.33
   557.9 2069.61   568.6 2069.26   664.1 2069.87   726.3 2066.77   759.8 2068.79
   766.1 2067.56   782.3 2060.15   809.3 2060.62   825.9 2057.26   842.5 2060.11
   853.9 2057.19   867.4 2050.85  1049.9 2050.87  1051.5 2051.03 1056.34  2057.3
  1068.6 2075.79  1091.4 2112.04  1099.7 2121.96  1116.3 2130.55  1129.1 2131.49
#Mann= 9 ,-1,0
       0      .1       0   358.4     .05       0   460.3     .08       0
   557.9     .05       0   568.6     .08       0   664.1      .1       0
   853.9    .035       0 1056.34    .025       0  1068.6      .1       0
Bank Sta=853.9,1056.34
XS Rating Curve= 0 ,0
Exp/Cntr(USF)=0,0
Exp/Cntr=0.5,0.3

Type RM Length L Ch R = 1 ,74035   ,100,93.7,91.4
BEGIN DESCRIPTION:
structure xs 3
channel burned per survey points
END DESCRIPTION:
XS GIS Cut Line= 6
  2212879.829386417885.3480720332212886.95089782 417786.01576846
2213012.11136855417312.0278013472212999.04369516417127.213563492
2212943.03938066416751.9846563332212902.83889449416669.917308523
#Sta/Elev= 30
       0 2089.18    56.6 2085.46   153.5 2085.74   208.1 2083.72   266.1 2078.36
     320 2079.63   375.5 2078.94   412.5 2075.92   644.8  2068.6   805.5 2069.39
  889.37 2060.05     896 2057.85  906.52 2052.69  918.73 2050.16  957.92 2047.16
 1044.57 2048.83 1053.49 2051.33 1062.84 2058.06 1075.03    2061  1088.6 2075.75
  1100.7 2079.45  1112.8 2089.23  1135.4 2101.62  1141.2 2101.66  1155.7 2096.94
  1167.7 2096.46  1179.9 2099.68  1194.6 2097.32  1215.5 2098.64  1245.9 2095.14
#Mann= 6 ,-1,0
       0      .1       0     320    .016       0   375.5      .1       0
     896    .035       0 1062.84     .08       0  1135.4      .1       0
#XS Ineff= 3 ,-1
   160.9  342.31 2084.06  342.31     763 2079.48  1105.9  1245.9 2080.21
Permanent Ineff=
       F       F       F
Bank Sta=896,1062.84
XS Rating Curve= 0 ,0
Exp/Cntr(USF)=0,0
Exp/Cntr=0.5,0.3

Type RM Length L Ch R = 3 ,74000   ,,,
BEGIN DESCRIPTION:
Bridge No.: 54075GRL030 Greenbrier River Trail
JV notes: road deck updated per surveyed XS data points
channel burned per surveyed cross sections
structure opening based on survey data, photos, and aerial imagery
square nose pier per photos provided by survey and data provided in survey data viewer
surveyed inverts are 7-8' below inverts from lidar:
 surveyed invert US is 2047.23
 surveyed invert DS is 2047.14
END DESCRIPTION:
Bridge Culvert--1,0,-1,-1, 0
Deck Dist Width WeirC Skew NumUp NumDn MinLoCord MaxHiCord MaxSubmerge Is_Ogee
31,12,2.6,0, 375, 375, , , 0.98, 0, 0,0,,
   61.25  62.433  64.878  66.698  69.131  70.595  71.685  73.454   75.83  76.312
  79.171  81.658  82.528  84.888  87.747  89.227  91.632  93.464  95.925  96.618
  99.181  102.04 102.624 104.898 106.592 107.757 109.322 111.578 113.474 116.021
 119.191 122.719 124.909 126.538 127.767 129.418 131.525 133.485 136.117 139.202
 142.815 144.919 146.485 147.778 149.514 150.636 153.495 156.212 159.212 161.445
 162.911 164.929 167.788 169.609 171.419 173.505 176.405 179.222 181.392 183.006
  184.94 186.484 189.021 190.606 192.252 193.434 194.572 196.263 200.123 201.921
  203.79  204.75 205.674 207.579 209.559 210.408 211.225 213.237 215.328 216.066
 216.777 221.097 224.553 227.879 230.211 232.634 235.869 238.403 241.527 244.532
 247.185 249.941 252.842  255.71   258.5 261.478 264.158 267.301  269.85 271.717
 272.718 274.119 275.585 276.633 278.453 281.001 281.548 284.188 286.464 287.883
  292.79 294.764 296.295 298.525 300.122 301.646  304.26 308.528 309.995 311.042
 312.862  315.41 318.597 322.292 325.789  335.62 338.669 341.536 344.432 347.407
 350.382 351.565 353.357 356.332 358.756  360.39 362.281 365.256 369.215 371.206
 372.218  374.18 375.324  378.04  380.13 381.193 386.865 389.054 395.691 397.979
 399.142 404.516 406.903 409.878 411.842 413.341 417.061 418.883 421.356 421.995
 423.718 425.107  428.22 429.888 431.332 435.227 440.669 443.781 446.735 453.118
 455.484 458.243 459.342 462.455 465.567 468.282 469.751 471.792 478.016 481.128
 484.241 485.346 487.478  490.64 494.479 499.243 503.543 505.125 508.765 510.354
  514.52 516.446 518.687 519.672 522.773  527.02  529.35 531.187 532.576 535.354
 537.336  539.52 542.253 543.687 547.854 548.705  551.93 555.156 556.187 560.354
  564.52 565.908 568.059 571.611 574.052 576.731  580.75 584.769 588.788 591.866
 593.582 597.244 600.845 601.519 608.883 612.902 616.921  623.04 626.538 628.978
 632.997 637.016 641.019 644.683 645.342 649.022 653.154 661.088 664.871 669.028
 676.589 681.031 684.401 689.034 693.035 697.036   702.1 703.931 709.995 713.046
 720.582 724.777 725.316 730.318  732.25  759.23  797.23  797.23     798  924.59
  970.22  1071.9  1071.9 1072.47 1104.97 1136.661139.8041143.9311147.6851151.151
1152.6181156.9621160.3061163.3581165.6491169.4621175.5651178.6171181.6691184.721
1186.3681187.772  1193.9 1198.99 1199.981201.4321203.0011208.3361210.218 1211.96
 1213.751214.9461217.3671217.9321220.9181222.6731223.9051226.8911229.8771232.863
1235.4311236.6681238.8361241.8221244.8091247.7951250.7811253.4941253.9021256.754
 1259.741262.5261263.1181265.7121268.6991271.5571274.6711280.589 1283.631285.132
1286.6161289.6211292.5891295.5751298.6521301.5481302.9781307.2011310.5061311.901
1316.7151320.8241324.9011328.1611330.7961333.849 1335.941339.5381341.0831343.988
1345.226 1348.071350.9141356.7121359.4471361.6591365.1361366.8031369.4361370.824
1371.9461373.6681375.7981379.357 1382.161385.0561390.765 1393.621396.475 1399.33
1402.0021405.0391407.3451410.7491413.6041415.2331416.4591419.3141422.4111425.023
1427.8781432.4551433.5881437.4771438.601
2080.5712080.5582080.5882080.6312080.6572080.6352080.6492080.6322080.6362080.625
2080.6332080.6752080.6822080.6452080.6632080.6892080.6852080.6712080.706  2080.7
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                                                 2076.98 2076.98 2076.98  2076.9
 2076.87  2076.8  2076.8
      15  16.183  18.628  20.448  22.881  24.345  25.435  27.204   29.58  30.062
  32.921  35.408  36.278  38.638  41.497  42.977  45.382  47.214  49.675  50.368
  52.931   55.79  56.374  58.648  60.342  61.507  63.072  65.328  67.224  69.771
  72.941  76.469  78.659  80.288  81.517  83.168  85.275  87.235  89.867  92.952
  96.565  98.669 100.235 101.528 103.264 104.386 107.245 109.962 112.962 115.195
 116.661 118.679 121.538 123.359 125.169 127.255 130.155 132.972 135.142 136.756
  138.69 140.234 142.771 144.356 146.002 147.184 148.322 150.013 153.873 155.671
  157.54   158.5 159.424 161.329 163.309 164.158 164.975 166.987 169.078 169.816
 170.527 174.847 178.303 181.629 183.961 186.384 189.619 192.153 195.277 198.282
 200.935 203.691 206.592  209.46  212.25 215.228 217.908 221.051   223.6 225.467
 226.468 227.869 229.335 230.383 232.203 234.751 235.298 237.938 240.214 241.633
  246.54 248.514 250.045 252.275 253.872 255.396  258.01 262.278 263.745 264.792
 266.612  269.16 272.347 276.042 279.539  289.37 292.419 295.286 298.182 301.157
 304.132 305.315 307.107 310.082 312.506  314.14 316.031 319.006 322.965 324.956
 325.968  327.93 329.074  331.79  333.88 334.943 340.615 342.804 349.441 351.729
 352.892 358.266 360.653 363.628 365.592 367.091 370.811 372.633 375.106 375.745
 377.468 378.857  381.97 383.638 385.082 388.977 394.419 397.531 400.485 406.868
 409.234 411.993 413.092 416.205 419.317 422.032 423.501 425.542 431.766 434.878
 437.991 439.096 441.228  444.39 448.229 452.993 457.293 458.875 462.515 464.104
  468.27 470.196 472.437 473.422 476.523  480.77   483.1 484.937 486.326 489.104
 491.086  493.27 496.003 497.437 501.604 502.455  505.68 508.906 509.937 514.104
  518.27 519.658 521.809 525.361 527.802 530.481   534.5 538.519 542.538 545.616
 547.332 550.994 554.595 555.269 562.633 566.652 570.671  576.79 580.288 582.728
 586.747 590.766 594.769 598.433 599.092 602.772 606.904 614.838 618.621 622.778
 630.339 634.781 638.151 642.784 646.785 650.786  655.85 657.681 663.745 666.796
 674.332 678.527 679.066 684.068     686  712.98  750.98  750.98  751.75  878.34
  923.97 1025.65 1025.65 1026.22 1058.72 1090.411093.5541097.6811101.4351104.901
1106.3681110.7121114.0561117.1081119.3991123.2121129.3151132.3671135.4191138.471
1140.1181141.522 1147.65 1152.74 1153.731155.1821156.7511162.0861163.968 1165.71
  1167.51168.6961171.1171171.6821174.6681176.4231177.6551180.6411183.6271186.613
1189.1811190.4181192.5861195.5721198.5591201.5451204.5311207.2441207.6521210.504
 1213.491216.2761216.8681219.4621222.4491225.3071228.4211234.339 1237.381238.882
1240.3661243.3711246.3391249.3251252.4021255.2981256.7281260.9511264.2561265.651
1270.4651274.5741278.6511281.9111284.5461287.599 1289.691293.2881294.8331297.738
1298.976 1301.821304.6641310.4621313.1971315.4091318.8861320.5531323.1861324.574
1325.6961327.4181329.5481333.107 1335.911338.8061344.515 1347.371350.225 1353.08
1355.7521358.7891361.0951364.4991367.3541368.9831370.2091373.0641376.1611378.773
1381.6281386.2051387.3381391.2271392.351
2080.5712080.5582080.5882080.6312080.6572080.6352080.6492080.6322080.6362080.625
2080.6332080.6752080.6822080.6452080.6632080.6892080.6852080.6712080.706  2080.7
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                                                 2076.98 2076.98 2076.98  2076.9
 2076.87  2076.8  2076.8
Pier Skew, UpSta & Num, DnSta & Num=  ,938.34, 2 ,893.34, 2 , 0 , 0 , 0 ,,
       9       9
       0    2077
       9       9
       0    2077
BR Coef=-1 ,-1 , 0 ,, 0 ,,,0.8,0,2,0,
WSPro=,,,, 1 ,,,, 0 ,,,, 0 ,,,,-1 ,-1 ,-1 , 0 , 0 , 0 , 0 , 0
BR U #Sta/Elev= 398
       0 2089.18     4.2 2088.47     8.4 2087.99    12.2 2087.73    20.2 2087.49
    28.2 2087.12    32.3    2087    36.3 2086.63    40.3 2086.46    44.3 2086.23
    48.3  2085.9    52.3 2085.62    56.6 2085.46    60.4 2085.47    64.6 2085.62
    68.3 2085.51    72.4 2085.28    81.9 2085.16    82.8 2085.18    84.4 2085.14
    88.4 2084.94    92.4 2085.05    96.4 2085.22   100.5 2085.25   107.8 2085.16
   112.9 2085.24   117.6 2085.17   125.3 2085.34   133.6 2085.29   133.9  2085.3
   135.1 2085.32   137.2 2085.39   141.9 2085.39     147 2085.58   153.5 2085.74
   154.3 2085.73   158.4 2085.46     167 2085.19   169.8 2085.07     175 2084.97
   179.6  2084.7   187.4 2084.42   192.7 2083.92   195.7 2083.73   199.9 2083.76
   208.1 2083.72   212.3  2083.5   215.5 2083.11   216.4 2083.05   222.1 2082.99
   224.7    2083   228.9 2082.83   231.8 2082.31   241.6  2080.9   244.9 2080.27
   245.4 2080.15   248.2 2079.69   249.6 2079.39   253.7 2078.85     262 2078.49
   264.5 2078.44   266.1 2078.36     269 2078.36   270.3 2078.35   274.3 2078.63
   282.7 2079.07   284.1 2079.05   286.8 2079.05     291 2079.09   291.6 2079.12
   293.9 2079.24   295.1  2079.3     303 2079.18   303.4 2079.18   307.6 2079.15
   310.2 2079.19   315.8 2079.35     320 2079.63   323.3 2079.72   324.1 2079.76
   325.6  2079.8   332.4 2079.92   340.7 2079.94   349.4 2079.84   350.9 2079.82
   353.1 2079.77   353.9 2079.75   361.4 2079.63   362.4 2079.56   365.3 2079.52
   365.5  2079.5   365.7  2079.5   366.3 2079.48     369 2079.34   375.5 2078.94
   376.6 2078.91     378 2078.84   381.7 2078.58   382.1 2078.55   385.3 2078.24
   390.4 2078.12   391.8 2078.01   395.1 2077.65   397.1 2077.36   398.3  2077.2
   398.7 2077.16   399.3 2077.12   402.8  2076.9   404.9  2076.7   404.9 2076.69
     407 2076.43   408.1 2076.34   410.6 2076.05   411.1    2076   411.4 2075.99
   412.5 2075.92   417.9 2075.84   423.5 2075.56     431 2075.48   431.8 2075.45
   433.3 2075.36   434.2 2075.32     436 2075.19   437.5 2075.14   438.9 2075.07
   440.1 2075.02   443.3 2074.96   452.5 2075.05   456.7 2074.89   457.1 2074.88
   469.1 2074.61   472.7 2074.81   473.2 2074.83   473.5 2074.83   474.7  2074.8
   477.3 2074.69   480.1 2074.53   481.4 2074.46   483.4 2074.41   483.7 2074.41
   485.6 2074.39   489.7 2074.25   496.6 2073.91   497.9 2073.83   502.1 2073.72
   509.8 2073.39   511.2 2073.34   513.1 2073.28   516.4 2073.17   519.7 2073.08
   522.2 2073.03   522.7 2073.01     523    2073   524.1 2072.94   526.3 2072.83
   526.8 2072.82   530.9 2072.53   532.9 2072.44     535 2072.33   542.8 2072.09
   552.7 2071.68   555.2 2071.58   555.7 2071.55   557.1 2071.45   559.8 2071.27
   560.7 2071.24   562.6 2071.15     568 2071.03   569.1    2071   572.4 2070.87
   573.6 2070.82   575.7 2070.73   576.3  2070.7   577.2 2070.65     579  2070.5
   588.9 2070.14   589.8 2070.07   592.4 2069.89   592.7 2069.88     593 2069.87
   596.2 2069.83   596.7 2069.82   599.9 2069.86   600.7 2069.86   601.6 2069.84
   603.7 2069.81   610.2 2069.56   611.2  2069.5   612.7 2069.41   637.4 2068.85
   640.4 2068.85   640.8 2068.84   641.1 2068.83   644.8  2068.6   644.9  2068.6
   645.6 2068.59   648.8 2068.57   649.1 2068.57   652.8 2068.68   653.4 2068.69
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BR U #Mann= 6
       0      .1     320    .016   375.5      .1     896     .03 1062.84     .08
  1135.4      .1
BR D #Sta/Elev= 454
       0 2086.62     6.9 2086.54    19.4 2087.48    23.5  2087.9    27.7 2087.93
      36 2087.47    40.1 2087.42    44.3 2087.53    47.4 2087.45    52.6 2087.39
    58.3 2087.49    60.4 2087.49    66.8 2087.33    73.4 2087.22    81.7 2086.95
    85.9 2086.87    94.2 2086.34    99.2 2086.24   106.7 2085.95   123.3 2085.72
   131.6 2085.38   141.3 2084.81   148.3  2084.3   152.4 2084.22   156.6 2084.31
   157.5 2084.29   169.1 2083.85   173.7 2083.58   177.4  2083.5   181.5 2083.37
   185.7 2083.35     194 2082.89   202.3 2082.92   206.5 2082.31   210.6 2081.63
   214.8 2081.23     219 2080.91   222.3 2080.42   223.1 2080.34   227.3 2080.11
     232 2080.02   233.8 2080.04   238.4 2079.99   243.9 2079.88   248.1 2079.62
   252.2 2079.49   254.6 2079.63   256.4 2079.71   260.5 2079.54   264.3 2079.33
   264.7 2079.32   265.4 2079.29   267.6 2079.19   268.9 2079.14     273 2078.89
     277 2078.81   277.3  2078.8   280.5 2078.78   281.3  2078.8   282.8 2078.72
   283.8 2078.66   285.5  2078.6     287 2078.37   289.7 2078.04   293.5 2077.66
     298 2077.08   300.2 2076.87   303.2 2076.61     306 2076.27   306.3 2076.25
   306.4 2076.23     307 2076.17   309.7 2075.96   310.5 2075.88   311.8 2075.84
   312.9 2075.85   314.6 2075.75   316.2 2075.73   317.6 2075.53   318.8 2075.46
   321.6 2075.16   322.6 2075.14   325.9  2074.9   331.2 2074.38   332.3 2074.32
   335.1 2074.13   335.4 2074.11   338.8 2074.25   343.7 2074.22   345.3 2074.18
   346.7 2074.11   352.5 2074.02   356.2 2074.06   358.2 2074.18   358.3 2074.18
   360.4 2074.33   364.1 2074.44   364.5 2074.45   368.7 2074.12   372.8 2074.16
   377.7 2073.91   380.7 2073.83   381.1 2073.81   384.3 2073.68   385.2 2073.63
   389.4 2073.72   394.1 2073.99   397.6 2074.14   401.8 2074.07   403.7 2073.94
   403.9 2073.92   405.9 2073.79   418.3 2073.52   422.5 2073.32   426.6 2072.97
   426.8 2072.97   430.1 2073.07   430.7 2073.05   431.8    2073   433.4 2072.98
   434.9 2072.88   436.7 2072.89   437.4 2072.92   443.2 2073.04   446.5 2073.21
   447.3 2073.18   449.8 2072.94   451.4 2072.81   455.6  2072.4   456.3  2072.4
   459.1 2072.23   459.6 2072.22   459.7 2072.21   471.1 2072.49   472.1 2072.51
   472.7  2072.5   474.8 2072.46   475.9 2072.44   476.2 2072.43   476.8 2072.44
   479.2  2072.5   480.4 2072.52   484.5 2073.08   488.7 2073.55     489 2073.49
   492.8 2073.09   496.9 2072.36   501.1 2071.95   504.9 2071.99   505.2 2071.99
   505.4 2072.01   506.2 2072.05   508.7 2072.11   513.5  2072.4   521.8 2072.09
     525 2071.78   525.9 2071.72   528.3 2071.26     530    2071   531.6 2070.73
   534.2 2070.32   534.9 2070.24   537.5 2069.81   538.1 2069.71   538.3 2069.69
   542.4  2069.4   544.2 2069.46   546.6 2069.56   547.8 2069.77     548  2069.8
   554.6 2071.12   555.6 2071.11   557.8  2070.9   558.6 2070.88   559.4 2070.72
     562 2069.92   563.2 2069.73   566.2  2069.4   566.6 2069.36     567 2069.38
   570.5 2069.64   570.6 2069.65   570.8 2069.66     574 2069.85   574.6 2069.89
   574.7 2069.89   578.7 2069.44   582.2 2068.98   582.7 2068.92   583.1 2068.88
     586 2068.56   590.7 2068.12   591.6 2068.14   593.6 2068.26   594.7 2068.28
   595.8 2068.53   597.4 2068.92   598.7  2069.2   600.1 2069.24   601.2 2069.25
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BR D #Mann= 4
       0      .1   809.1     .03  1012.6     .08  1094.1      .1
BC Design=,, 0 ,, 0 ,,,,,,
BC Use User HTab Curves=0
BC User HTab FreeFlow(D)= 0

Type RM Length L Ch R = 1 ,73941   ,555.1,448,352.7
BEGIN DESCRIPTION:
structure xs 2
channel burned per survey points
END DESCRIPTION:
XS GIS Cut Line= 6
2212940.23714062417811.7973229652213041.98033628417453.905398084
2213086.78378788417284.025644096 2213096.1178403417108.545458658
2213032.64628387416751.9846563332212965.44110646416613.840680563
#Sta/Elev= 30
       0 2086.62    60.4 2087.49   202.3 2082.92   223.1 2080.34   285.5  2078.6
   335.4 2074.11   459.7 2072.21   488.7 2073.55   542.4  2069.4   554.6 2071.12
   590.7 2068.12   602.7  2069.3   638.7 2067.45   650.8 2068.71   682.8 2065.49
   710.1 2066.07   783.8 2062.34     800 2060.54   809.1 2056.61  819.49 2053.94
  839.21 2052.14  916.61 2047.14  993.01 2052.81  1007.2  2054.5  1012.6 2056.79
  1035.7  2081.5    1056 2096.76  1068.2 2099.11  1094.1 2097.42  1239.3 2084.63
#Mann= 4 ,-1,0
       0      .1       0   809.1    .035       0  1012.6     .08       0
  1094.1      .1       0
#XS Ineff= 2 , 0
           733.6  2076.6    1043          2079.9
Permanent Ineff=
       F       F
Bank Sta=809.1,1012.6
XS Rating Curve= 0 ,0
Exp/Cntr(USF)=0,0
Exp/Cntr=0.5,0.3

Type RM Length L Ch R = 1 ,73493   ,549.8,336.3,137.4
BEGIN DESCRIPTION:
xs 1 - channel burned 9.73':
lidar invert = 2054.23
effective invert = 2044.50
END DESCRIPTION:
XS GIS Cut Line= 3
2213822.30711833417058.1415756072213340.67001362416583.971712829
2213004.64412661416606.373438629
#Sta/Elev= 30
       0 2097.85    36.7 2093.28    47.4 2088.87    53.5 2087.78    64.1 2088.18
    81.4 2086.85   106.8 2082.14   149.6 2077.62     186 2070.45   211.5 2067.06
   252.2 2065.91     275 2067.45   311.7 2066.58   349.2 2068.06   379.1 2063.93
   389.1  2060.3   395.4  2055.6   395.9 2055.33  400.01 2045.05   400.5 2044.69
   648.5  2044.5   654.1 2055.31   669.7 2062.66   680.4 2065.17   736.5 2070.31
     809 2075.32   887.9 2078.68   937.1 2081.04   988.7  2081.4  1012.7 2081.24
#Mann= 5 ,-1,0
       0      .1       0   395.4    .035       0   654.1     .05       0
   887.9     .06       0   988.7      .1       0
#XS Ineff= 2 , 0
          344.11 2080.55
Permanent Ineff=
       F       F
#Block Obstruct= 1 ,-1
  898.68  936.59 2091.29
Bank Sta=395.4,654.1
XS Rating Curve= 0 ,0
Exp/Cntr(USF)=0,0
Exp/Cntr=0.3,0.1

Type RM Length L Ch R = 1 ,73157   ,627.5,518.5,287.4
BEGIN DESCRIPTION:
channel burned 7.33':
lidar invert = 2054.06
interpolated invert = 2046.73
END DESCRIPTION:
Node Name=D
XS GIS Cut Line= 3
 2213792.4381506416191.9415113192213050.84600112 416538.25631377
2212995.69543642416596.883045016
#Sta/Elev= 30
       0 2236.77    31.2 2214.18    75.3 2174.08   145.6 2119.02   163.6 2102.12
   178.7 2089.38   184.7 2085.74   194.5 2083.12   199.7 2079.37   203.4 2075.96
   213.3 2063.89223.89992056.335   231.8 2047.08   232.8  2046.8   420.4 2046.73
   446.2 2046.73452.69982055.868   459.4 2058.79   485.6  2062.7   503.6 2062.57
   521.2 2065.65   556.5 2067.33   658.1 2071.79   715.5 2071.26   759.6 2072.54
     797 2074.65   815.9 2077.29   851.6 2077.67   866.4 2080.41     899 2080.95
#Mann= 4 ,-1,0
       0      .1       0223.8999    .035       0452.6998      .1       0
   556.5     .05       0
#Block Obstruct= 1 ,-1
  666.35  728.93 2091.87
Bank Sta=223.8999,452.6998
XS Rating Curve= 0 ,0
Exp/Cntr(USF)=0,0
Exp/Cntr=0.3,0.1

Type RM Length L Ch R = 1 ,72638   ,361.5,352.6,325.4
BEGIN DESCRIPTION:
channel burned 3.25':
lidar invert = 2053.75
effective invert = 2050.50
END DESCRIPTION:
XS GIS Cut Line= 3
2213159.58939674415665.5009550062212916.29028666416497.535505445
2212912.88139126416561.895348612
#Sta/Elev= 30
       0 2376.14    24.7 2354.83    47.6 2331.46      67 2317.03    87.2 2298.08
   128.3 2266.76   154.7 2248.93     196 2211.99   203.9 2203.13   216.4 2179.96
     233 2162.38   245.5  2144.5   253.9 2134.76   266.4 2115.05   274.7  2099.1
   278.9 2092.82   299.7  2079.9   312.2 2066.75   316.4 2063.77   328.2 2058.78
341.19942056.157   349.7  2050.5   528.9  2050.5 536.9992055.828   553.9 2066.31
   562.3 2068.09   573.2 2068.04   670.6 2070.04   816.5 2070.03   931.3 2080.57
#Mann= 4 ,-1,0
       0      .1       0341.1994    .035       0 536.999      .1       0
   573.2     .05       0
Bank Sta=341.1994,536.999
XS Rating Curve= 0 ,0
Exp/Cntr(USF)=0,0
Exp/Cntr=0.3,0.1

Type RM Length L Ch R = 1 ,72286   ,554.5,527.2,453.2
BEGIN DESCRIPTION:
channel burned 2.71':
lidar invert = 2053.47
interpolated invert = 2050.76
END DESCRIPTION:
XS GIS Cut Line= 2
2212763.82557426415631.898366305 2212590.2121993416600.773007179
#Sta/Elev= 30
       0 2338.57    21.6 2326.72    58.2 2294.56    86.6 2275.02   127.3 2229.68
   160.4 2187.76   176.6 2174.65   200.4 2147.32   224.8 2125.91   249.2 2090.21
   261.4 2078.75   277.6 2073.34   285.8 2064.06   300.6  2056.2   314.2 2050.79
   407.7 2050.76   497.1 2050.76   503.9 2055.91   513.3 2061.45   541.8 2068.66
   670.4 2066.86   740.9 2068.04     749 2070.32   761.2 2077.79   781.5 2077.11
   793.7 2070.95   834.4 2072.48   850.6  2077.1     940 2092.36   984.3 2101.74
#Mann= 8 ,-1,0
       0      .1       0   300.6    .035       0   503.9      .1       0
   541.8     .05       0   670.4      .1       0   761.2    .016       0
   781.5      .1       0     940     .05       0
#XS Ineff= 2 , 0
                          764.51         2098.17
Permanent Ineff=
       F       F
Bank Sta=300.6,503.9
XS Rating Curve= 0 ,0
Exp/Cntr(USF)=0,0
Exp/Cntr=0.3,0.1

Type RM Length L Ch R = 1 ,71758   ,511.1,463.8,351.6
BEGIN DESCRIPTION:
channel burned 2.38':
lidar invert = 2053.06
interpolated invert = 2050.68
END DESCRIPTION:
XS GIS Cut Line= 3
 2212242.9854494415628.1647453382212158.97897764415818.579414643
2212211.24967118416537.301450744
#Sta/Elev= 30
       0  2182.5    57.9 2158.42   114.8 2137.16   158.5 2118.07   189.1 2101.65
   197.1 2094.42   210.7 2079.33   218.7 2072.42   226.6 2069.59   242.8 2067.58
   254.8 2061.29   262.9 2054.74   266.9 2050.71   511.5 2050.68   515.5 2054.84
   527.6 2062.51   531.6 2063.85   551.3 2065.43   600.5 2066.21     676 2064.61
     750 2066.08   768.2 2066.96   787.4 2076.35   804.3 2076.15   820.3 2069.29
   844.4 2069.25   852.4 2070.98   864.5 2077.32   896.5 2083.95   928.7 2095.01
#Mann= 7 ,-1,0
       0      .1       0   262.9    .035       0   515.5      .1       0
   551.3     .05       0     750      .1       0   787.4    .016       0
   804.3      .1       0
#XS Ineff= 2 , 0
                          790.99         2088.27
Permanent Ineff=
       F       F
Bank Sta=262.9,515.5
XS Rating Curve= 0 ,0
Exp/Cntr(USF)=0,0
Exp/Cntr=0.3,0.1

Type RM Length L Ch R = 1 ,71294   ,492.2,491.7,417.5
BEGIN DESCRIPTION:
channel burned 2.49':
lidar invert = 2052.66
interpolated invert = 2050.17
END DESCRIPTION:
XS GIS Cut Line= 2
2211578.40091731415770.0423420752211933.09490915416600.773007179
#Sta/Elev= 30
       0 2245.78    68.7 2191.93    90.4 2171.74   146.8 2126.67   151.3 2119.29
     160 2099.48   164.3 2092.34   168.7 2086.77   180.5 2075.73   186.6 2071.89
   203.5 2068.06   217.1  2060.6   238.4 2058.27     249 2054.49   255.7 2050.17
   507.9 2050.25   513.8 2054.36   525.3 2060.21   564.6 2062.69   607.2 2061.61
   640.1 2063.43   741.3 2065.67   777.9 2067.88   799.3 2075.46   799.3 2075.47
   814.5 2075.75   825.4  2075.5   834.1 2077.53   860.2  2092.1   903.3 2112.15
#Mann= 7 ,-1,0
       0      .1       0     249    .035       0   513.8      .1       0
   640.1     .05       0   741.3      .1       0   799.3    .016       0
   814.5      .1       0
Bank Sta=249,513.8
XS Rating Curve= 0 ,0
Exp/Cntr(USF)=0,0
Exp/Cntr=0.3,0.1
