HEC-RAS study GRNBRRRV.prj: GRNBRRRV

--- GRNBRRRV.g01 (geometry) --- (continued)

Type RM Length L Ch R = 1 ,70803   ,134.9,405.6,504.2
BEGIN DESCRIPTION:
channel burned 2.32':
lidar invert = 2052.22
effective invert = 2049.90
END DESCRIPTION:
XS GIS Cut Line= 3
2211177.03666339 415811.112172712211182.63709484416201.275563736
2211606.40307456416759.451898266
#Sta/Elev= 30
       0 2204.51    78.1 2152.45   146.1 2096.02   178.1 2071.89   185.6 2068.48
   226.1 2063.84   246.1 2055.34   258.1 2053.39   326.1 2053.15   342.1 2057.26
   358.1 2057.66   475.5 2052.77   570.9 2053.25   575.9 2050.28     591  2049.9
   670.6 2049.96   805.2 2049.95  807.98 2050.28   809.5 2053.02     822 2057.43
   876.5 2060.44   907.4 2066.44   927.5 2067.47   942.5 2073.65   952.6 2075.24
   962.6 2075.35   977.7 2074.75   997.8 2082.64  1027.9 2097.53    1091 2133.42
#Mann= 6 ,-1,0
       0      .1       0   570.9     .08       0   670.6    .035       0
   809.5      .1       0   952.6    .016       0   962.6      .1       0
Bank Sta=570.9,809.5
XS Rating Curve= 0 ,0
Exp/Cntr(USF)=0,0
Exp/Cntr=0.3,0.1

Type RM Length L Ch R = 1 ,70397   ,287.7,335.9,354.7
BEGIN DESCRIPTION:
channel burned 4.31':
lidar invert = 2051.54
interpolated invert = 2047.23
END DESCRIPTION:
XS GIS Cut Line= 2
2211068.76165535415829.7802775432210960.48664731 416893.86225307
#Sta/Elev= 30
       0 2173.48    19.5 2166.57    31.6 2159.43    99.9 2111.37     120 2093.87
   144.1 2077.45   172.3 2066.79   204.4 2063.78   240.6 2063.51   272.8 2056.84
   325.4 2053.63   546.2 2051.09   582.4  2055.4   606.5 2056.21   642.3  2052.9
   654.8 2047.23   839.7 2047.37     843 2052.92   851.8 2063.21   855.8 2065.98
   871.9 2067.45   890.4 2073.16   901.4 2073.77   908.1 2074.42   940.2 2090.94
  1004.6 2132.76  1016.6 2144.63  1032.7 2146.15  1044.8 2158.98  1069.6 2176.98
#Mann= 5 ,-1,0
       0      .1       0   642.3    .035       0     843      .1       0
   890.4    .016       0   901.4      .1       0
Bank Sta=642.3,843
XS Rating Curve= 0 ,0
Exp/Cntr(USF)=0,0
Exp/Cntr=0.3,0.1

Type RM Length L Ch R = 1 ,70061   ,461.9,518.5,557.6
BEGIN DESCRIPTION:
channel burned 3.58':
lidar invert = 2050.99
interpolated invert = 2047.41
END DESCRIPTION:
Node Name=C
XS GIS Cut Line= 2
2210797.99367338415843.614173445 2210571.2694113416950.306379033
#Sta/Elev= 30
       0 2138.28    42.4 2126.91    54.7 2118.46      74 2099.88    83.3 2093.18
    95.5 2087.93   124.1 2067.74   144.5 2062.14   226.2 2063.74   332.3 2061.66
   381.3 2062.77   446.7 2057.74   461.8 2052.56   471.2 2047.41   818.2 2047.65
   826.2 2052.63   846.8 2062.16   895.8 2064.53     908 2067.02   920.3 2072.15
   940.7 2072.91   948.9 2075.74   993.8 2102.04  1022.4 2120.22  1046.6  2138.7
  1063.2 2141.73  1079.5 2156.83  1112.2 2177.91  1120.4 2187.54  1129.7 2195.27
#Mann= 5 ,-1,0
       0      .1       0   461.8    .035       0   826.2      .1       0
   920.3    .016       0   940.7      .1       0
#Block Obstruct= 1 ,-1
  860.84  889.44 2081.02
Bank Sta=461.8,826.2
XS Rating Curve= 0 ,0
Exp/Cntr=0.3,0.1

Type RM Length L Ch R = 1 ,69543   ,386,451.7,486.5
BEGIN DESCRIPTION:
channel burned 3.58':
lidar invert = 2050.52
interpolated invert = 2046.94
END DESCRIPTION:
XS GIS Cut Line= 2
2210375.69153628415748.592415378 2209999.4088226416846.225725801
#Sta/Elev= 30
       0 2107.61    69.4    2088    97.9  2075.6   110.6    2066   123.2  2063.9
   135.9 2058.07   144.4 2056.56   448.8 2058.74   499.6 2058.14   529.2 2053.33
   560.6 2051.76   571.5 2046.94   840.9 2046.98  846.51 2050.78   863.9 2051.64
   875.9 2054.95   909.8 2056.87   968.9  2055.7   994.3 2053.15  1011.2 2057.75
  1028.1 2057.08  1045.1 2059.12  1058.1 2069.05  1066.2 2070.81  1074.7 2071.01
  1083.1 2074.51    1100 2090.23  1138.1 2115.83  1150.8  2125.9  1160.3 2135.93
#Mann= 5 ,-1,0
       0      .1       0   560.6    .035       0   863.9      .1       0
  1066.2    .016       0  1074.7      .1       0
#Block Obstruct= 1 ,-1
  911.85  958.14 2073.21
Bank Sta=560.6,863.9
XS Rating Curve= 0 ,0
Exp/Cntr=0.3,0.1

Type RM Length L Ch R = 1 ,69091   ,544.9,488,451.9
BEGIN DESCRIPTION:
channel burned 2.74'
lidar invert = 2049.66
interpolated invert = 2046.92
END DESCRIPTION:
XS GIS Cut Line= 3
  2210084.694629415575.5176048952209612.64947831416442.094116092
2209554.59710483416765.885806404
#Sta/Elev= 30
       0 2097.81    34.5 2088.46      93    2080   129.4 2064.43   143.1 2061.42
   226.9 2058.23   243.3 2061.44   279.7 2057.67   293.5 2053.97   308.3 2053.64
   393.6 2057.97   434.6 2056.18   586.4 2059.97   603.1 2057.69   617.9  2051.4
   625.9 2046.92   921.6 2046.92   933.3 2051.59   945.2 2056.56   967.5 2059.66
  1071.2 2056.91  1087.5 2053.75  1180.9 2059.14  1189.1 2060.46  1209.4 2070.05
  1220.7 2070.16  1225.6 2070.47  1241.9  2081.4    1297 2107.43  1315.8 2114.88
#Mann= 6 ,-1,0
       0      .1       0   617.9    .035       0   933.3      .1       0
  1209.4    .016       0  1220.7      .1       0    1297     .06       0
#XS Ineff= 2 , 0
             240 2070.23
Permanent Ineff=
       F       F
#Block Obstruct= 1 ,-1
 1036.38 1077.74 2075.38
Bank Sta=617.9,933.3
XS Rating Curve= 0 ,0
Exp/Cntr=0.3,0.1

Type RM Length L Ch R = 1 ,68603   ,349,332.5,284.9
BEGIN DESCRIPTION:
channel burned 2.21':
lidar invert = 2048.58
interpolated effective invert = 2046.37
END DESCRIPTION:
XS GIS Cut Line= 3
2209359.49598359415355.7134059752209445.23928549415593.527546993
2209053.30500144416761.134325226
#Sta/Elev= 30
       0 2095.58   259.7 2071.79   300.7 2056.94   328.4 2049.37   349.5 2048.66
   367.1 2052.47   395.5 2053.87   430.3 2053.68   446.5 2049.81   450.7 2046.37
   847.4  2046.6   868.5 2049.98   923.8 2055.07   972.6  2054.9  1003.5 2061.14
  1025.4 2060.29  1121.6  2056.2  1163.1 2056.74  1185.3 2056.93  1218.7 2053.45
  1265.1 2056.09  1294.6 2067.94  1307.3 2068.05  1345.2 2090.22  1368.4 2106.38
    1378  2106.8  1383.2 2108.62  1396.9 2122.47    1417 2135.03  1484.4 2186.28
#Mann= 9 ,-1,0
       0      .1       0   446.5    .035       0   868.5     .07       0
  1025.4     .06       0  1163.1      .1       0  1294.6    .016       0
  1307.3      .1       0  1368.4    .016       0    1378      .1       0
#Block Obstruct= 1 ,-1
 1021.58 1093.32 2078.25
Bank Sta=446.5,868.5
XS Rating Curve= 0 ,0
Exp/Cntr=0.3,0.1

Type RM Length L Ch R = 1 ,68270   ,208.5,178.6,110.8
BEGIN DESCRIPTION:
channel burned 2.33':
lidar invert = 2047.81
interpolated effective invert = 2045.48
END DESCRIPTION:
XS GIS Cut Line= 3
 2209179.3951161415268.4199613012208872.96152506416319.801985021
2208846.51628224416718.651489928
#Sta/Elev= 30
       0  2091.9      83  2089.2   138.7 2068.93   187.1 2062.26   203.2 2065.65
   280.7 2061.46   300.8 2065.68   396.2 2051.14   492.4 2048.96   500.8 2045.48
   642.4 2045.55   650.8 2051.01     713  2054.3   763.2 2049.37     771 2045.59
   846.6  2048.8   931.3 2055.17     942 2059.17   983.6 2059.99  1136.6 2054.75
  1236.8 2056.32    1301 2056.48    1325  2068.3  1336.2 2067.39    1349 2067.78
  1370.5 2083.98  1381.1 2084.09    1413 2118.05  1460.7 2160.29  1494.9 2182.15
#Mann= 13 ,-1,0
       0      .1       0   492.4    .035       0   650.8      .1       0
   763.2    .035       0   846.6     .06       0   931.3     .05       0
   983.6     .06       0  1136.6     .05       0  1236.8     .07       0
  1336.2    .016       0    1349      .1       0  1370.5    .016       0
  1381.1      .1       0
#XS Ineff= 2 , 0
          310.04 2070.84
Permanent Ineff=
       F       F
#Block Obstruct= 1 ,-1
  995.64 1057.19 2075.36
Bank Sta=492.4,846.6
XS Rating Curve= 0 ,0
Exp/Cntr=0.3,0.1

Type RM Length L Ch R = 1 ,68092   ,679.4,658.3,647.9
BEGIN DESCRIPTION:
channel burned 2.30':
lidar invert = 2047.41
interpolated effective invert = 2045.11
END DESCRIPTION:
XS GIS Cut Line= 3
2208751.76849297415263.5488799212208865.19865978415621.885088695
2208705.36524291416787.122256794
#Sta/Elev= 30
       0 2094.84   341.6  2076.9   391.3 2071.96   419.6 2054.98   447.2 2049.49
   455.9 2045.11   613.4 2045.28   621.8 2049.96   637.6 2054.26   657.8 2054.94
   681.5 2049.39   690.1 2045.23   782.9 2045.29  799.49 2048.27   855.5 2053.79
   867.7 2057.32   944.4 2059.09  1017.1    2058  1146.3 2056.22  1158.4 2053.82
  1216.1 2055.51  1279.5 2058.85  1295.7 2066.07  1314.4 2067.41  1333.1 2067.56
  1340.1 2068.84  1372.4 2099.69  1400.7 2116.93  1494.5 2135.52    1552 2152.33
#Mann= 12 ,-1,0
       0     .08       0   341.6      .1       0   447.2    .035       0
   621.8      .1       0   681.5    .035       0  799.49     .06       0
   855.5     .08       0   944.4     .06       0  1017.1     .05       0
  1216.1     .07       0  1314.4    .016       0  1333.1      .1       0
#Block Obstruct= 2 ,-1
  960.72 1031.62 2074.54 1234.55 1254.75  2071.9
Bank Sta=447.2,799.49
XS Rating Curve= 0 ,0
Exp/Cntr(USF)=0,0
Exp/Cntr=0.3,0.1

Type RM Length L Ch R = 1 ,67434   ,304.6,292.3,224.2
BEGIN DESCRIPTION:
channel burned 2.67':
lidar invert = 2046.97
interpolated effective invert = 2044.30
END DESCRIPTION:
XS GIS Cut Line= 5
 2208432.8014794415225.2693369032208181.67852327415556.491856627
2208192.50278862415931.0114377532208129.72204959416032.759532047
2208103.74381275416649.742657023
#Sta/Elev= 30
       0 2096.55    65.1  2093.9   346.2 2066.42   464.4 2063.31   476.4 2052.94
   492.1 2049.48   508.4  2044.3   736.5 2044.33   743.5 2049.39   756.5 2055.81
   772.5 2056.55   806.7 2055.22   818.3 2048.45   830.5 2047.76   844.6 2047.54
     854 2052.91   885.2 2052.59   902.6 2055.91   942.3 2052.49    1009 2052.68
  1046.2 2055.59  1142.3 2059.57  1161.5 2059.42  1234.5 2060.06  1334.7 2058.94
  1354.7 2059.23  1374.7 2065.44  1390.7 2067.01  1454.8 2112.24  1527.4 2166.59
#Mann= 10 ,-1,0
       0      .1       0   492.1    .035       0   743.5      .1       0
   830.5     .06       0   942.3      .1       0  1046.2     .05       0
  1142.3     .06       0  1161.5     .05       0  1234.5     .06       0
  1334.7      .1       0
Bank Sta=492.1,743.5
XS Rating Curve= 0 ,0
Exp/Cntr(USF)=0,0
Exp/Cntr=0.3,0.1

Type RM Length L Ch R = 1 ,67141   ,628.7,722.3,756.6
BEGIN DESCRIPTION:
channel burned 4.39':
lidar invert = 2046.84
interpolated effective invert = 2042.45
END DESCRIPTION:
XS GIS Cut Line= 4
2208019.86215373414855.2369687682207903.62020026415088.247713038
2207893.55476783415310.5441101612207899.23186176416626.463599761
#Sta/Elev= 30
       0  2114.1    33.5 2103.82    79.9 2094.77   189.9 2086.08   313.4 2067.22
   357.4 2064.13   545.6 2062.62   585.6 2061.97   601.6 2061.72   753.6 2061.06
   769.6 2061.21   785.6 2058.72  808.56 2049.44   813.6 2047.13   817.6 2042.45
  1045.8 2042.49  1057.6 2049.19  1065.5 2050.86  1077.5 2051.09  1089.6 2053.78
  1133.4 2052.61  1229.6 2058.64  1253.6 2059.19  1573.6 2057.98  1623.3 2060.47
  1637.6 2065.57  1657.6 2068.31  1681.6 2087.71  1701.6 2101.18  1798.9 2174.85
#Mann= 15 ,-1,0
       0     .06       0    33.5     .07       0   357.4     .05       0
   545.6     .06       0   585.6    .016       0   601.6     .05       0
   753.6      .1       0  808.56    .035       0  1057.6     .06       0
  1065.5    .016       0  1077.5     .08       0  1133.4     .05       0
  1229.6    .016       0  1253.6     .05       0  1623.3      .1       0
#XS Ineff= 2 , 0
          539.19 2065.18
Permanent Ineff=
       F       F
#Block Obstruct= 3 ,-1
  108.21  178.39 2108.26  495.47  531.04 2078.41  668.06  705.82 2076.81
Bank Sta=808.56,1057.6
XS Rating Curve= 0 ,0
Exp/Cntr(USF)=0,0
Exp/Cntr=0.3,0.1

Type RM Length L Ch R = 1 ,66419   ,440.8,574.2,614.5
BEGIN DESCRIPTION:
channel burned 4.48':
lidar invert = 2046.53
interpolated effective invert = 2042.05
END DESCRIPTION:
XS GIS Cut Line= 3
2207810.86545032414547.5057629792207189.80606962415446.971072959
2207130.91250766 416619.48835204
#Sta/Elev= 30
       0 2137.14    60.4 2115.49   123.6 2103.84     143 2095.06   158.4 2094.71
   201.3 2087.22   296.4  2081.7   335.6 2078.74   612.7 2068.67   680.6  2061.2
   760.3 2059.05  1214.9 2061.22  1231.4 2060.47  1239.4 2051.74  1245.4 2048.64
  1255.5 2042.05  1543.8 2042.11  1550.5 2048.48  1559.8 2055.04    1581 2056.72
    1604 2057.31  1748.1 2054.68  1903.3 2057.36  1939.5 2059.33  1976.4 2066.14
  2000.4 2066.12  2008.4 2069.26  2038.6 2093.31  2136.6 2144.81    2267 2245.54
#Mann= 10 ,-1,0
       0      .1       0   296.4     .08       0   335.6     .06       0
   760.3     .05       0  1214.9      .1       0  1245.4    .035       0
  1550.5     .06       0    1581    .016       0    1604     .05       0
  1903.3      .1       0
#Block Obstruct= 3 ,-1
  850.52  900.88 2074.93 1098.11 1136.43 2075.61 1623.67 1693.49 2072.61
Bank Sta=1245.4,1550.5
XS Rating Curve= 0 ,0
Exp/Cntr(USF)=0,0
Exp/Cntr=0.3,0.1

Type RM Length L Ch R = 1 ,65845   ,322.5,500.6,600.5
BEGIN DESCRIPTION:
channel burned 4.98':
lidar invert = 2046.28
interpolated effective invert = 2041.30
END DESCRIPTION:
XS GIS Cut Line= 3
2207521.75160068414344.0552761982206654.41005178415366.661670282
2206493.79124642416437.453705972
#Sta/Elev= 30
       0 2153.78    85.4 2110.22   153.6 2092.49   200.3 2086.93   484.4 2066.11
   521.3 2066.45   535.5 2070.54   612.1 2063.38   725.3 2059.19  1359.6 2059.78
  1448.6 2061.07  1463.8 2061.02  1492.8 2060.67  1509.3 2049.02  1513.3 2041.95
  1517.4  2041.3  1824.8 2041.36  1830.4 2042.39  1832.9  2048.4  1844.5 2053.05
  1855.1 2053.53  1942.1 2055.52  2014.9 2057.46  2041.5  2065.1  2067.5 2066.51
  2152.4 2122.47  2358.7 2290.42  2366.8 2298.33  2382.9 2328.03  2423.7 2356.07
#Mann= 12 ,-1,0
       0     .06       0   153.6      .1       0   200.3     .05       0
  1359.6     .06       0  1448.6     .05       0  1463.8     .06       0
  1509.3    .035       0  1832.9     .06       0  1844.5    .016       0
  1855.1     .06       0  1942.1     .05       0  2041.5      .1       0
#Block Obstruct= 2 ,-1
 1429.84 1475.68 2076.41 1927.46 1981.82 2071.28
Bank Sta=1509.3,1832.9
XS Rating Curve= 0 ,0
Exp/Cntr(USF)=0,0
Exp/Cntr=0.3,0.1

Type RM Length L Ch R = 1 ,65344   ,324.6,608.9,691.6
BEGIN DESCRIPTION:
channel burned 6.29':
lidar invert = 2046.09
interpolated effective invert = 2039.80
END DESCRIPTION:
XS GIS Cut Line= 2
2207146.97438819414258.3919133432205915.56354715415805.686404915
#Sta/Elev= 30
       0 2103.84   257.3 2086.99   397.2 2073.98   460.6 2070.13   555.7 2058.49
     842 2057.12  1184.5 2057.56  1295.6 2059.38  1385.6 2060.35    1392 2058.21
  1398.8 2051.45  1417.7 2049.04  1427.3 2047.34  1430.5 2040.32    1435  2039.8
  1719.6 2039.88  1723.3 2040.41 1724.91 2044.83  1727.7  2047.5    1749 2053.03
    1757 2053.01    1771 2053.83  1787.7 2064.41  1811.6 2065.72  1817.3 2067.67
  1871.4 2110.89  1905.5 2141.98  1915.5 2147.94  1936.8 2153.58  1977.5 2156.36
#Mann= 7 ,-1,0
       0     .05       0  1295.6     .06       0  1417.7      .1       0
  1427.3    .035       0  1727.7      .1       0    1749    .016       0
    1757      .1       0
#Block Obstruct= 1 ,-1
 1340.01 1373.75 2074.23
Bank Sta=1427.3,1727.7
XS Rating Curve= 0 ,0
Exp/Cntr(USF)=0,0
Exp/Cntr=0.3,0.1

Type RM Length L Ch R = 1 ,64735   ,443.3,474.2,505
BEGIN DESCRIPTION:
channel burned 3.34':
lidar invert = 2045.84
interpolated effective invert = 2042.50
END DESCRIPTION:
Node Name=B
XS GIS Cut Line= 3
2206906.04618016 414129.896869062206611.57837035414568.921603693
2205294.50416645415259.582466713
#Sta/Elev= 30
       0 2102.08    96.7 2093.67   352.5 2077.96   456.3 2064.29   528.6 2060.13
     799 2054.78  1060.9 2056.37  1128.7 2058.54  1169.3 2050.12  1192.1 2051.06
  1203.9 2047.62    1210  2042.5  1494.5  2042.5 1501.36 2047.59  1512.6 2050.96
  1577.2 2049.35  1589.1 2049.27  1618.7 2052.73  1643.6 2054.46  1706.8 2053.66
  1734.3 2054.91  1746.1 2057.01  1760.9 2063.31  1797.1 2066.11  1801.6 2068.89
  1810.7 2078.58  1815.2 2080.83  1849.8 2087.74    1918 2096.04  2015.8 2103.48
#Mann= 8 ,-1,0
       0     .05       0  1060.9     .06       0  1169.3      .1       0
  1203.9    .035       0 1501.36      .1       0  1577.2    .016       0
  1589.1     .08       0  1618.7      .1       0
#Block Obstruct= 1 ,-1
 1659.97 1691.45 2071.15
Bank Sta=1203.9,1501.36
XS Rating Curve= 0 ,0
Exp/Cntr(USF)=0,0
Exp/Cntr=0.3,0.1

Type RM Length L Ch R = 1 ,64261   ,447.5,529.7,560
BEGIN DESCRIPTION:
channel burned 3.24':
lidar invert = 2045.64
interpolated effective invert = 2042.40
END DESCRIPTION:
XS GIS Cut Line= 2
2206777.55113588414113.8349885252205117.82348056414734.894369225
#Sta/Elev= 30
       0 2094.21   163.8 2081.14   402.9 2068.91   443.3 2068.12   622.1 2059.34
   781.5  2056.3   880.1 2057.34   902.6 2056.09   919.7 2046.28     924  2045.5
   932.5 2045.87   949.6 2050.18     971 2049.95   982.7 2047.98   988.9  2042.4
  1312.6 2042.42  1320.6 2047.79  1340.1  2048.7  1358.7 2050.95    1368 2051.09
  1440.8 2054.25  1496.3  2059.4  1513.4 2063.32  1530.4 2064.24  1564.6 2082.93
  1615.9 2118.54  1641.5 2129.86  1669.5 2133.78  1752.5 2135.96  1772.1 2138.03
#Mann= 8 ,-1,0
       0     .05       0   781.5     .06       0   880.1      .1       0
   982.7    .035       0  1320.6     .06       0  1340.1      .1       0
  1358.7    .016       0    1368      .1       0
#Block Obstruct= 3 ,-1
  195.47  228.12 2096.72  820.81  855.67 2073.19 1424.62  1459.8 2072.86
Bank Sta=982.7,1320.6
XS Rating Curve= 0 ,0
Exp/Cntr(USF)=0,0
Exp/Cntr=0.3,0.1

Type RM Length L Ch R = 1 ,63731   ,516.9,563,580
BEGIN DESCRIPTION:
channel burned 2.42':
lidar invert = 2043.64
interpolated effective invert = 2041.22
END DESCRIPTION:
XS GIS Cut Line= 2
2206638.34817124413797.9513379962205074.99179913414113.834988525
#Sta/Elev= 30
       0 2085.75   161.4 2077.16     243 2070.44   625.8 2056.43   634.7 2056.36
   717.5 2054.29   866.9 2056.02   882.42044.935   883.7 2041.63   891.8 2041.22
   997.9 2041.33  1006.1 2045.82  1026.1  2045.9  1030.6 2041.61  1034.7 2041.33
  1234.6 2041.33  1238.7 2041.78  1240.3 2044.46    1251 2045.08  1275.4 2051.18
  1311.6 2052.27  1397.9 2054.57  1410.1  2060.2  1410.1 2060.22  1418.3 2062.47
  1426.4 2062.53  1434.6 2062.93    1455 2072.59    1557 2134.16    1595 2141.62
#Mann= 12 ,-1,0
       0     .05       0   625.8    .016       0   634.7     .05       0
   717.5      .1       0   882.4    .035       0  1006.1      .1       0
  1026.1    .035       0    1251     .08       0  1311.6     .06       0
  1410.1      .1       0  1418.3    .016       0  1426.4      .1       0
#Block Obstruct= 2 ,-1
  719.75   773.7 2069.53 1308.07 1336.87 2068.94
Bank Sta=882.4,1251
XS Rating Curve= 0 ,0
Exp/Cntr(USF)=0,0
Exp/Cntr=0.3,0.1

Type RM Length L Ch R = 1 ,63168   ,372.9,428.9,453.3
BEGIN DESCRIPTION:
channel burned 5.47':
lidar invert = 2042.97
interpolated effective invert = 2037.50
END DESCRIPTION:
XS GIS Cut Line= 2
2206713.30361374413326.8028422932204957.20467521413519.545408717
#Sta/Elev= 30
       0 2133.77    81.6 2091.36   121.9 2074.07   129.9 2074.03   178.2  2065.5
   230.5 2060.88   415.6 2056.95   744.4 2053.42   902.6 2054.56   950.8 2051.07
   970.9 2052.86  1083.6 2054.53 1102.96 2043.96  1111.8 2037.62  1115.8  2037.5
  1377.4 2037.53  1381.1 2037.74  1388.2 2044.11  1397.5 2048.89  1421.6 2052.99
  1471.7 2052.87    1482 2052.88  1518.2 2052.76  1534.3 2059.78  1561.6 2061.94
  1578.6 2063.06  1610.7 2088.17  1660.3 2121.83  1699.3 2137.95  1766.6 2142.41
#Mann= 11 ,-1,0
       0      .1       0   121.9    .016       0   129.9     .06       0
   178.2     .05       0   970.9      .1       0 1102.96    .035       0
  1388.2     .06       0  1471.7    .016       0    1482     .06       0
  1561.6      .1       0  1660.3     .05       0
#XS Ineff= 2 , 0
          413.08 2079.07
Permanent Ineff=
       F       F
#Block Obstruct= 2 ,-1
  975.56 1021.36  2067.8 1431.39 1465.13 2068.15
Bank Sta=1102.96,1388.2
XS Rating Curve= 0 ,0
Exp/Cntr(USF)=0,0
Exp/Cntr=0.3,0.1

Type RM Length L Ch R = 1 ,62740   ,456.8,557.5,605.5
BEGIN DESCRIPTION:
channel burned 4.88':
lidar invert = 2042.38
interpolated effective invert = 2037.50
END DESCRIPTION:
XS GIS Cut Line= 2
2206665.11797213413037.6889926562204871.54131235413032.335032478
#Sta/Elev= 30
       0 2148.06    44.9 2124.91   112.8 2100.02     157 2078.79   184.9 2070.27
   192.9 2070.78   213.1 2070.87   264.9  2060.7   316.9 2056.57   736.9 2053.67
   912.9 2055.57  1012.9 2050.37  1036.9 2053.26 1070.23 2043.96  1078.2 2037.96
  1084.9  2037.5  1344.9  2037.5  1348.9 2037.71 1354.88 2044.04  1372.9 2049.99
  1469.1 2054.51  1484.9 2059.53  1528.9 2057.06  1600.7 2077.83    1661 2094.97
    1681 2095.06    1689 2094.69  1708.4 2108.72  1748.2 2125.64  1793.6 2137.36
#Mann= 10 ,-1,0
       0      .1       0   192.9    .016       0   213.1      .1       0
   736.9     .06       0  1012.9      .1       0 1070.23    .035       0
 1354.88      .1       0  1600.7     .06       0    1661    .016       0
    1681      .1       0
#Block Obstruct= 3 ,-1
  900.63   935.4  2070.3 1393.13 1431.55 2067.91 1621.19 1646.43 2104.86
Bank Sta=1070.23,1354.88
XS Rating Curve= 0 ,0
Exp/Cntr(USF)=0,0
Exp/Cntr=0.3,0.1

Type RM Length L Ch R = 1 ,62182   ,405,408.3,410.1
BEGIN DESCRIPTION:
channel burned 3.74':
lidar invert = 2041.54
interpolated effective invert = 2037.80
END DESCRIPTION:
XS GIS Cut Line= 2
 2206649.0560916412721.8053421282204657.38290521412288.134567673
#Sta/Elev= 30
       0 2153.64    59.3 2111.63   119.6 2078.86   140.1 2071.11   185.1 2062.99
   209.7 2062.56   279.3 2054.83   389.8 2053.98   520.8 2053.84   627.2 2051.72
     835 2053.71     922 2051.42   950.6 2043.56   958.8  2037.8  1224.9 2037.85
  1253.6 2043.71  1278.1 2050.48  1310.9 2051.47  1322.4 2055.16  1343.6 2059.78
  1351.8 2059.88  1425.5 2065.46  1454.2 2065.36  1470.5 2065.55  1621.6  2073.5
  1687.5 2076.94  1740.7 2072.87  1834.9 2095.28  1920.6 2108.83  2038.3 2114.23
#Mann= 16 ,-1,0
       0      .1       0   185.1    .016       0   209.7      .1       0
   389.8     .06       0   520.8     .07       0   627.2     .06       0
     835      .1       0   950.6    .035       0  1253.6     .07       0
  1322.4     .05       0  1343.6    .016       0  1351.8     .06       0
  1425.5     .07       0  1454.2    .016       0  1470.5     .05       0
  1621.6      .1       0
#Block Obstruct= 4 ,-1
  452.75   486.3 2071.03  535.01  564.23 2069.93 1290.45 1318.99  2069.9
 1547.49 1571.56 2087.13
Bank Sta=950.6,1253.6
XS Rating Curve= 0 ,0
Exp/Cntr(USF)=0,0
Exp/Cntr=0.3,0.1

Type RM Length L Ch R = 1 ,61774   ,515.2,500.5,517.6
BEGIN DESCRIPTION:
channel burned 3.71':
lidar invert = 2040.91
interpolated effective invert = 2037.20
END DESCRIPTION:
XS GIS Cut Line= 2
2206638.34817124412309.550408387  2204710.922507411875.879633932
#Sta/Elev= 30
       0 2199.56    47.3 2164.06     158  2094.5   209.6 2069.78   260.5 2055.14
   272.8 2055.03   293.3 2051.28   346.6 2051.63   493.7 2053.57   502.4 2054.08
   666.4 2049.24   674.6 2050.59   801.7 2053.85   826.3 2043.56   838.6  2037.2
  1117.4 2037.27  1123.9 2043.18  1154.3 2047.63  1174.8 2058.23  1195.3 2058.91
  1203.5 2058.89  1215.8 2063.38  1314.1 2066.46  1495.9 2070.19  1502.8 2070.59
  1615.9 2075.37  1679.1 2079.16  1769.4 2086.98  1822.6 2112.16  1975.6 2127.91
#Mann= 17 ,-1,0
       0      .1       0   260.5    .016       0   272.8      .1       0
   346.6     .06       0   493.7    .016       0   502.4     .06       0
   666.4    .016       0   674.6      .1       0   826.3    .035       0
  1123.9     .08       0  1195.3    .016       0  1203.5     .05       0
  1314.1     .07       0  1495.9    .016       0  1502.8     .05       0
  1615.9     .06       0  1679.1      .1       0
#Block Obstruct= 5 ,-1
   555.3  584.19 2070.61  747.46  787.84 2069.76 1288.67    1380 2082.97
 1454.43 1488.73 2085.71  1532.3 1558.67 2087.96
Bank Sta=826.3,1123.9
XS Rating Curve= 0 ,0
Exp/Cntr(USF)=0,0
Exp/Cntr=0.3,0.1

Type RM Length L Ch R = 1 ,61273   ,250.6,223.4,197.1
BEGIN DESCRIPTION:
structure xs 4 - channel burned 4.12':
lidar invert = 2040.31
interpolated effective invert = 2036.19
END DESCRIPTION:
XS GIS Cut Line= 3
2206635.69616405411693.6484684412206060.34523783411669.845410933
2205080.09358779411446.426173911
#Sta/Elev= 30
       0 2236.26   215.7 2105.35   331.8 2050.38   347.8 2050.53   399.9 2045.78
   423.9 2047.04   451.9 2050.25     524 2048.16     568 2053.28   613.3 2051.31
   629.4 2047.05   638.9 2043.71   649.9 2036.19   900.1 2036.19   904.2 2036.65
   907.3 2043.88   917.3 2056.54   928.8 2061.04     974 2063.92   998.6 2057.82
  1017.6 2058.18  1027.3 2062.05    1056 2064.99  1124.5 2066.28  1311.6 2071.25
  1375.1 2074.18  1382.9 2074.71  1428.5 2077.46  1532.1 2085.91  1581.2 2086.83
#Mann= 14 ,-1,0
       0      .1       0   331.8    .016       0   347.8      .1       0
   423.9     .06       0   629.4      .1       0   638.9    .035       0
   907.3     .08       0   998.6    .016       0  1017.6     .06       0
  1124.5      .1       0  1311.6     .07       0  1375.1    .016       0
  1382.9     .06       0  1428.5      .1       0
#XS Ineff= 2 , 0
                          967.21         2077.85
Permanent Ineff=
       F       F
#Block Obstruct= 1 ,-1
 1068.24 1093.36 2081.08
Bank Sta=638.9,907.3
XS Rating Curve= 0 ,0
Exp/Cntr(USF)=0,0
Exp/Cntr=0.5,0.3

Type RM Length L Ch R = 1 ,61050   ,83.3,86.3,83.4
BEGIN DESCRIPTION:
structure xs 3
END DESCRIPTION:
XS GIS Cut Line= 2
2206594.08162848411449.9389071842205108.19545397411362.120575357
#Sta/Elev= 30
       0 2222.13   102.1  2159.2   205.6 2093.15   250.3 2067.41   266.4 2054.47
   278.7 2053.49   370.6 2050.62   454.7 2051.98   498.8 2051.85  526.54 2047.69
  537.63 2042.84  550.46 2038.15  562.51 2037.09  733.44 2035.57  801.55 2037.86
   814.6 2042.97   836.1 2054.85   838.6 2053.55   851.4 2057.93   899.2 2058.39
   935.5 2058.93  1007.7 2063.93  1141.3 2068.03    1266 2073.95  1276.1 2074.41
  1288.2 2074.21  1340.2 2079.14  1394.8 2085.32  1452.4 2102.87  1488.5 2106.18
#Mann= 12 ,-1,0
       0      .1       0   266.4    .016       0   278.7     .06       0
   454.7     .07       0  537.63    .035       0   814.6      .1       0
   899.2    .016       0   935.5     .06       0  1141.3     .07       0
    1266    .016       0  1276.1      .1       0  1340.2      .1       0
#XS Ineff= 2 , 0
          502.93 2050.69  856.47         2059.06
Permanent Ineff=
       F       F
#Block Obstruct= 2 ,-1
 1210.58 1242.61    2092  1314.1 1336.94 2098.92
Bank Sta=537.63,814.6
XS Rating Curve= 0 ,0
Exp/Cntr(USF)=0,0
Exp/Cntr=0.5,0.3

Type RM Length L Ch R = 3 ,61022   ,,,
BEGIN DESCRIPTION:
Bridge No.: 54075GRL020 Seebert River Rd (Rte 27/3)
JV notes: road deck updated per surveyed XS data points
channel burned per surveyed cross sections
structure opening based on survey data, photos, and aerial imagery
surveyed inverts are 5-6' below inverts from lidar:
 surveyed invert US is 2035.6
 surveyed invert DS is 2035.1
END DESCRIPTION:
Bridge Culvert--1,0,-1,-1, 0
Deck Dist Width WeirC Skew NumUp NumDn MinLoCord MaxHiCord MaxSubmerge Is_Ogee
20,16,2.6,0, 430, 430, , , 0.98, 0, 0,0,,
      -7  -5.263  -4.801  -4.379  -1.066   -.551   3.131   7.106   7.328  10.934
  11.525  14.762  15.723   18.59   19.92  22.419  23.229  24.117  26.247  27.233
  28.314  30.075  31.237  32.511  33.903  35.241  36.709  37.731  39.246   43.25
  45.103  45.388  47.254  51.258  53.044  53.497  55.263  59.267  63.271  64.529
  66.089  67.275  68.357  70.286  71.279  75.284  78.681  79.842  83.292  87.075
  87.498  91.326  95.305  98.983  99.667 102.811 107.317 111.322 115.326  119.33
 121.952 123.334  125.78 129.047 129.609 131.343 135.347 139.351 141.093 141.639
 143.355 144.922 145.836  147.36  148.75 150.033 151.364 155.368 158.427 159.372
 160.234 162.625 163.377 164.063 166.822 167.381 167.891 171.385 175.216 179.413
 183.204 183.611 187.032 187.808  190.86 192.005 194.688  195.41 199.415 200.399
 202.345 203.419 204.597 206.173 207.423 208.794 210.001 211.427 215.432 217.188
 217.658 219.436  223.44 225.314 225.583 227.444 231.448  232.97 233.977 235.453
 236.799 238.174 239.457 240.627 242.371 243.461 244.455 246.569 247.465 248.283
 250.766  251.47 255.474  255.94  259.16 259.768 263.482 263.596 267.486 271.253
 271.491 271.752 275.081 275.949 279.499 283.503 284.343 286.565 291.512 295.516
  299.52 301.878 303.524 307.529 311.533 315.537 319.541 321.019 322.118 323.546
  327.55 331.554 332.504  334.71 338.907 340.161 343.567 347.571 355.579 359.302
  363.13  364.09 366.958 367.592 371.596 375.601 378.443 382.271 385.076 386.099
 387.613 389.273 389.927 391.617 395.622 399.626  403.63  405.24 406.062 407.634
 411.639 414.457 415.643 416.725 420.553 422.851 423.651 427.656 431.245 435.443
  439.64 443.837 447.351 451.681 452.231 455.007 456.444     459  488.54  520.63
  522.93  523.83  582.37  614.91  646.28  675.65  710.13  761.94  774.08  836.47
  836.47   839.6  870.31  915.75 917.411 924.084 928.515 932.523 935.393 936.531
 940.539 942.931 948.555  950.47  954.24 958.009 960.579 964.587 968.595 980.611
 984.395 991.934 993.447 995.703 996.6511000.6591006.2831007.0121008.6751010.562
1014.5511016.6911020.6991024.7071028.7151031.9561033.3981036.7311040.5141044.064
1052.7631056.7711057.6291059.7841063.2761064.8611073.0271076.831 1080.221081.193
1085.2761089.3591090.3871093.4431095.4031097.1651101.6091105.6921107.3311108.342
 1110.721113.858 1119.281120.5571122.1861123.7851126.3511129.2961131.015 1133.47
1134.681 1143.651147.1761149.6121156.0681158.0041159.6711163.8361165.7531168.001
1168.9811172.3591180.4961184.6611186.7131188.3511191.5791192.9911194.8071197.156
1198.0361201.2641204.4921205.4861207.7211209.6511215.4211217.9811220.6341222.146
1224.8951229.7761234.6411236.7751239.9161242.8831251.5371255.0181257.5881259.064
1261.0621264.6191275.2441279.2891282.1961283.3341285.7121287.3671291.3711295.374
1299.3781301.7421303.3811304.8911305.9171307.3841308.7361310.0931311.3881315.391
1318.444 1320.271322.6191324.115 1327.961331.805 1335.651341.523 1343.341343.496
1347.1851347.6721351.4221354.8751356.023 1358.721360.1981364.374 1366.411367.435
1370.2551371.4391372.725  1374.1  1376.91379.4451383.4491387.4521391.4561395.459
1399.4621401.0141401.9531403.4661404.8591406.1281407.4691408.7041410.3041411.473
1415.4761419.4791424.0841427.0061427.9291431.181 1431.491435.6191439.4641443.309
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  2052.72052.7362053.3962053.7632054.1162054.4472054.836 2055.422055.557 2056.26
 2056.26
      13  14.737  15.199  15.621  18.934  19.449  23.131  27.106  27.328  30.934
  31.525  34.762  35.723   38.59   39.92  42.419  43.229  44.117  46.247  47.233
  48.314  50.075  51.237  52.511  53.903  55.241  56.709  57.731  59.246   63.25
  65.103  65.388  67.254  71.258  73.044  73.497  75.263  79.267  83.271  84.529
  86.089  87.275  88.357  90.286  91.279  95.284  98.681  99.842 103.292 107.075
 107.498 111.326 115.305 118.983 119.667 122.811 127.317 131.322 135.326  139.33
 141.952 143.334  145.78 149.047 149.609 151.343 155.347 159.351 161.093 161.639
 163.355 164.922 165.836  167.36  168.75 170.033 171.364 175.368 178.427 179.372
 180.234 182.625 183.377 184.063 186.822 187.381 187.891 191.385 195.216 199.413
 203.204 203.611 207.032 207.808  210.86 212.005 214.688  215.41 219.415 220.399
 222.345 223.419 224.597 226.173 227.423 228.794 230.001 231.427 235.432 237.188
 237.658 239.436  243.44 245.314 245.583 247.444 251.448  252.97 253.977 255.453
 256.799 258.174 259.457 260.627 262.371 263.461 264.455 266.569 267.465 268.283
 270.766  271.47 275.474  275.94  279.16 279.768 283.482 283.596 287.486 291.253
 291.491 291.752 295.081 295.949 299.499 303.503 304.343 306.565 311.512 315.516
  319.52 321.878 323.524 327.529 331.533 335.537 339.541 341.019 342.118 343.546
  347.55 351.554 352.504  354.71 358.907 360.161 363.567 367.571 375.579 379.302
  383.13  384.09 386.958 387.592 391.596 395.601 398.443 402.271 405.076 406.099
 407.613 409.273 409.927 411.617 415.622 419.626  423.63  425.24 426.062 427.634
 431.639 434.457 435.643 436.725 440.553 442.851 443.651 447.656 451.245 455.443
  459.64 463.837 467.351 471.681 472.231 475.007 476.444     479  508.54  540.63
  542.93  543.83  602.37  634.91  666.28  695.65  730.13  781.94  794.08  856.47
  856.47   859.6  890.31  935.75 937.411 944.084 948.515 952.523 955.393 956.531
 960.539 962.931 968.555  970.47  974.24 978.009 980.579 984.587 988.5951000.611
1004.3951011.9341013.4471015.7031016.6511020.6591026.2831027.0121028.6751030.562
1034.5511036.6911040.6991044.7071048.7151051.9561053.3981056.7311060.5141064.064
1072.7631076.7711077.6291079.7841083.2761084.8611093.0271096.831 1100.221101.193
1105.2761109.3591110.3871113.4431115.4031117.1651121.6091125.6921127.3311128.342
 1130.721133.858 1139.281140.5571142.1861143.7851146.3511149.2961151.015 1153.47
1154.681 1163.651167.1761169.6121176.0681178.0041179.6711183.8361185.7531188.001
1188.9811192.3591200.4961204.6611206.7131208.3511211.5791212.9911214.8071217.156
1218.0361221.2641224.4921225.4861227.7211229.6511235.4211237.9811240.6341242.146
1244.8951249.7761254.6411256.7751259.9161262.8831271.5371275.0181277.5881279.064
1281.0621284.6191295.2441299.2891302.1961303.3341305.7121307.3671311.3711315.374
1319.3781321.7421323.3811324.8911325.9171327.3841328.7361330.0931331.3881335.391
1338.444 1340.271342.6191344.115 1347.961351.805 1355.651361.523 1363.341363.496
1367.1851367.6721371.4221374.8751376.023 1378.721380.1981384.374 1386.411387.435
1390.2551391.4391392.725  1394.1  1396.91399.4451403.4491407.4521411.4561415.459
1419.4621421.0141421.9531423.4661424.8591426.1281427.4691428.7041430.3041431.473
1435.4761439.4791444.0841447.0061447.9291451.181 1451.491455.6191459.4641463.309
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  2052.72052.7362053.3962053.7632054.1162054.4472054.836 2055.422055.557 2056.26
 2056.26
Pier Skew, UpSta & Num, DnSta & Num=  ,582.37, 2 ,619.99, 2 , 0 , 0 , 0 ,,
       3       3
       0  2056.5
       3       3
       0  2056.5
Pier Skew, UpSta & Num, DnSta & Num=  ,646.28, 2 ,683.76, 2 , 0 , 0 , 0 ,,
       3       3
       0  2056.5
       3       3
       0  2056.5
Pier Skew, UpSta & Num, DnSta & Num=  ,710.13, 2 ,747.61, 2 , 0 , 0 , 0 ,,
       3       3
       0  2056.5
       3       3
       0  2056.5
Pier Skew, UpSta & Num, DnSta & Num=  ,774.08, 2 ,811.67, 2 , 0 , 0 , 0 ,,
       3       3
       0  2056.5
       3       3
       0  2056.5
BR Coef=-1 ,-1 , 0 ,, 0 ,,,0.8,0,1.2,0,
WSPro=,,,, 1 ,,,, 0 ,,,, 0 ,,,,-1 ,-1 ,-1 , 0 , 0 , 0 , 0 , 0
BR U #Sta/Elev= 442
       0 2222.13     1.9 2221.02     5.9 2218.35    10.1  2215.7    17.9  2210.5
    21.9 2208.15      30    2203      38 2198.26      42 2195.58      50 2190.77
      54  2188.5      62 2183.29    65.1 2181.45      70 2178.44      74 2176.05
    78.2 2173.69      82 2171.45    86.1 2168.72    90.1 2166.27    94.9 2163.42
    99.2 2160.95   102.1  2159.2   106.1 2156.57   110.1 2154.08   114.1 2151.67
   122.1 2146.54   130.1 2141.28   134.1 2138.73   138.1 2136.29   142.2  2133.6
   142.5 2133.35     146 2130.83   150.1  2128.4   154.2 2126.12   157.6  2123.7
   170.2 2115.28   182.2  2107.8   186.2  2105.4   190.2 2102.86   195.5 2099.85
   198.3 2098.21     203 2094.85   205.6 2093.15   210.3 2090.32   218.3 2085.31
   222.3    2083   230.3 2078.25   234.3 2075.96   238.3 2073.91   242.3 2071.98
   250.3 2067.41   254.3 2064.83   258.4 2061.01   262.4 2056.93   266.4 2054.47
   270.4 2053.71   278.7 2053.49   282.3 2053.32   298.4 2052.23   305.2 2052.08
   310.4 2051.91   316.5 2051.62   341.9 2051.11   354.7 2051.05   358.5 2050.97
   362.5  2050.8   366.5 2050.77   370.6 2050.62   382.6 2050.57   384.6 2050.58
   386.6  2050.6   388.4 2050.71   388.8 2050.74   390.6 2050.85   394.6 2051.52
   397.3 2051.84   398.6 2051.98   402.6 2052.18   403.6 2052.17   406.6 2052.19
   410.6 2052.06   414.6 2051.76   418.6 2051.58   418.7 2051.58   419.7 2051.58
   422.5 2051.57   422.6 2051.57   426.3 2051.45   426.6 2051.43   434.7  2051.3
   442.7 2051.36   454.7 2051.98   456.5 2051.99   456.9 2051.98   462.7 2051.92
   474.7 2052.41   478.7 2052.31   482.5  2052.4   486.8 2052.38   490.6 2052.19
   494.8 2052.05   498.1 2051.88   498.8 2051.85   503.7 2051.16   505.7 2050.81
   510.8 2050.12   514.8 2049.38   516.5 2049.07   517.1 2049.02   518.8 2048.69
  526.54 2047.69  537.63 2042.84  543.97 2040.33  550.46 2038.15  562.51 2037.09
   606.1 2036.11  675.42  2035.6  733.44 2035.57  784.67  2037.1  801.55 2037.86
  807.54 2040.32   814.6 2042.97  823.24 2048.08   836.1 2054.85   838.6 2053.55
   839.4 2053.88   840.2 2054.27   842.4 2055.37   843.4 2055.82   848.7 2057.15
   851.4 2057.93     853    2058   853.8 2058.06   855.4 2058.13   857.2 2058.14
   857.6 2058.14   863.4 2058.22   865.7 2058.38   867.4  2058.5     870 2058.45
   874.2 2058.37   875.4 2058.33   879.4 2058.18   883.4 2058.25     884 2058.26
     887 2058.31   899.2 2058.39   899.5 2058.39   899.8 2058.39     903 2058.39
   903.5 2058.39   904.1 2058.37   906.7 2058.28   907.5 2058.26   908.3 2058.26
   910.5  2058.2   911.5  2058.2   914.3 2058.25   915.5 2058.29   916.8 2058.32
   918.1 2058.35   919.5 2058.38   921.1 2058.41   921.9 2058.42   927.5 2058.59
   935.5 2058.93     937 2058.94   939.5 2058.97   940.8 2058.95   942.4 2058.92
   943.6 2058.91   944.6    2059   947.6 2059.29   948.4  2059.5   950.9 2060.26
   951.6 2060.44   955.6 2061.03   959.4 2061.37   959.6 2061.38   959.7 2061.38
   962.1 2061.37   963.6 2061.35   971.6 2061.52   972.2 2061.49   974.8 2061.38
   975.6 2061.35   979.6 2061.54   980.7 2061.55   982.4 2061.53   983.6 2061.55
     985 2061.59   986.2 2061.64   987.6 2061.69   989.2 2061.76     990  2061.8
   991.6 2061.87   995.6  2062.2   997.6 2062.48   999.6 2062.81  1001.3 2063.12
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BR U #Mann= 12
       0      .1   266.4    .016   278.7     .06   454.7     .07  537.63     .03
   814.6      .1   899.2    .016   935.5     .06  1141.3     .07    1266    .016
  1276.1      .1  1340.2      .1
BR D #Sta/Elev= 441
       0 2247.12     5.1 2243.52    13.1 2238.05    17.1 2235.12    25.1 2229.79
    33.2 2224.13    37.2 2221.61    41.2 2218.99    45.2 2216.29    53.3 2211.09
    54.2 2210.47    57.3 2208.58    61.3 2205.97    65.3  2203.5    69.8 2200.45
    74.2 2197.35    76.3 2196.01    85.4 2189.94      92  2185.5    93.4 2184.51
   101.5 2179.34   113.5 2171.95   116.7 2169.92   124.1 2165.06   127.7 2162.64
   129.6 2161.44   133.6 2158.76   138.8 2155.38   153.5 2145.42   161.7 2139.64
   162.9 2138.91   169.8 2134.31   171.7 2133.12   173.8 2131.87   177.8 2129.29
   181.8 2126.46   185.8 2123.71   193.9 2118.34   207.2 2110.04   215.9 2104.42
     218 2103.17     222 2100.43   223.3 2099.61     226 2097.81     230 2095.33
     234  2092.7   238.1 2089.84   246.1 2084.84   250.1 2082.21   254.1 2079.76
   256.3 2078.33   266.2 2072.16   267.4 2071.45     271 2069.23   278.2 2065.14
   278.4 2065.07   282.3 2063.02   286.9 2060.84   290.3 2059.28   291.4 2058.69
   294.3 2057.06   298.3 2054.24   302.3 2053.12   306.4 2053.07   307.8    2053
   310.4 2052.89   318.4 2051.89   322.4 2051.54   322.4 2051.53   326.8 2051.34
   330.5 2051.24   350.6 2050.99   359.2 2050.57   370.2 2050.52   370.6 2050.52
   374.7 2050.67   378.7 2050.69   386.7 2050.61   390.7 2050.45   392.3 2050.42
   393.3 2050.41   394.7 2050.39   398.8 2050.55   402.1 2050.76   402.8  2050.8
   403.3 2050.85   406.6 2051.14   414.3 2051.96   430.9 2053.53   438.9 2054.25
     443 2054.42   443.7 2054.43   446.4 2054.44     447 2054.44     451 2054.35
   454.8 2053.91     455 2053.89     459 2053.73     463 2053.64   464.2 2053.64
   465.8 2053.61   467.1 2053.61   475.1  2053.9   477.5 2053.96   480.5    2054
   481.9 2053.99   483.1    2054   495.2 2053.69   503.2 2053.72   507.2 2053.68
   511.2 2053.44   515.3 2053.06   523.3 2052.72   527.3 2052.27   531.3 2051.63
     532  2051.5   534.8 2051.03   535.8 2050.81   539.7 2049.85   543.3 2048.78
   543.5 2048.74   547.3 2047.69   547.3 2047.68   551.1 2046.67   551.4  2046.6
   555.4 2044.69   569.6 2040.42  580.99 2037.64  598.56  2037.5  631.44 2036.46
  653.17 2036.22   695.3  2035.1  720.24  2035.6  759.22 2036.54  790.39 2036.36
  816.76  2037.4  823.07 2037.36   829.4 2040.18  842.24 2045.47   863.7 2049.32
   864.3  2049.5   867.3 2050.59   867.7 2050.72   868.1 2050.82   871.5 2051.83
   871.7 2051.88   879.7 2053.71   883.7 2054.45   884.2  2054.5   887.2 2054.85
   887.7 2054.91   888.4 2054.97     891 2055.19   891.8 2055.26   892.6 2055.36
   895.8 2055.77   896.8 2055.94   898.6 2056.23   899.8 2056.41   902.5 2056.93
   903.8 2057.19   906.3 2057.55   907.8 2057.77   910.1 2057.85   911.8 2057.92
   926.3 2057.96     933 2058.01   935.8 2058.05   936.8 2058.06   938.9 2058.09
   940.6 2058.12   943.1 2058.18   947.8 2058.23   948.3 2058.21   951.5 2058.05
   955.8 2057.97   955.9 2057.98   959.9 2058.42   963.8 2058.75   964.2 2058.79
   972.6  2059.8   975.9 2060.11   976.8  2060.2   978.8 2060.44   979.9 2060.54
     981 2060.67   982.6  2060.9   983.9 2061.04   985.2 2061.16   987.9 2061.41
   991.9 2061.68   995.9 2061.78   997.8 2061.82   999.9 2061.88  1013.2 2062.72
  1014.7 2062.83  1015.9 2062.91    1017 2062.99  1018.9 2063.13  1020.8 2063.26
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BR D #Mann= 12
       0      .1   290.3    .016   302.3     .06   465.8    .016   495.2     .07
   569.6     .03   829.4      .1   892.6    .016   948.3     .05    1080     .07
  1265.2    .016  1280.2      .1
BC Design=,, 0 ,, 0 ,,,,,,
BC Use User HTab Curves=0
BC User HTab FreeFlow(D)= 0

Type RM Length L Ch R = 1 ,60964   ,245.3,242.4,243.2
BEGIN DESCRIPTION:
structure xs 2
END DESCRIPTION:
XS GIS Cut Line= 3
2206629.20896121411383.1969749952206102.29897025411334.018709172
2205164.39918634411288.353176622
#Sta/Elev= 30
       0 2247.12    33.2 2224.13   193.9 2118.34   266.2 2072.16   290.3 2059.28
   302.3 2053.12   326.8 2051.34   394.7 2050.39   438.9 2054.25   465.8 2053.61
   495.2 2053.69   534.8 2051.03   569.6 2040.42  580.99 2037.64   695.3  2035.1
  823.07 2037.36   829.4 2040.18  842.24 2045.47   892.6 2055.36   907.8 2057.77
   948.3 2058.21    1080 2066.67    1100 2068.76  1265.2 2074.33  1280.2 2075.15
  1332.3 2077.26  1391.3 2084.49  1412.4 2090.09  1444.7 2102.26  1468.2 2106.62
#Mann= 12 ,-1,0
       0      .1       0   290.3    .016       0   302.3     .06       0
   465.8    .016       0   495.2     .07       0   569.6    .035       0
   829.4      .1       0   892.6    .016       0   948.3     .05       0
    1080     .07       0  1265.2    .016       0  1280.2      .1       0
#XS Ineff= 2 , 0
           535.6 2050.69   883.8          2057.8
Permanent Ineff=
       F       F
#Block Obstruct= 4 ,-1
  400.49  458.06 2073.77 1060.46 1086.01  2087.3 1153.13 1171.56 2090.87
 1197.92  1268.4 2094.59
Bank Sta=569.6,829.4
XS Rating Curve= 0 ,0
Exp/Cntr(USF)=0,0
Exp/Cntr=0.5,0.3

Type RM Length L Ch R = 1 ,60721   ,382.9,379.1,358.1
BEGIN DESCRIPTION:
structure xs 1 - channel burned 3.61':
lidar invert = 2039.75
interpolated effective invert = 2036.14
END DESCRIPTION:
Node Name=A
XS GIS Cut Line= 2
2206537.87789611411116.2292462412205231.14111853411045.974580779
#Sta/Elev= 30
       0 2182.32    57.8 2147.66   149.9 2083.62     194  2059.5   205.8 2051.06
     218 2051.54     230 2051.26   274.1    2047   289.6 2040.29   414.3 2040.11
   442.3 2043.17  458.02 2040.39   466.4 2036.14   746.8 2036.14   750.8 2039.97
   758.8 2046.18   774.8 2048.76   790.8 2056.86   806.6 2057.37   814.2 2057.36
   842.9 2054.68     907 2055.98  1080.3 2067.53  1118.3 2070.72  1128.9 2071.13
  1139.3 2073.93    1183 2076.79  1215.5 2083.14  1281.3 2105.87  1308.6 2110.67
#Mann= 12 ,-1,0
       0      .1       0     218    .016       0     230      .1       0
  458.02    .035       0   750.8     .08       0   806.6    .016       0
   814.2     .05       0  1080.3     .06       0  1118.3    .016       0
  1128.9     .06       0    1183     .05       0  1281.3      .1       0
#XS Ineff= 2 , 0
                           805.5         2069.33
Permanent Ineff=
       F       F
#Block Obstruct= 1 ,-1
 1013.97 1066.05 2082.74
Bank Sta=458.02,750.8
XS Rating Curve= 0 ,0
Exp/Cntr(USF)=0,0
Exp/Cntr=0.3,0.1

Type RM Length L Ch R = 1 ,60342   ,76.6,83.9,107.7
BEGIN DESCRIPTION:
location of decommissioned structure - cross section cut across old deck location to capture area and mannings update to reflect conditions
remains of low watercourse crossing added as blocked obstructions - elevation assumed as 10yr WSEL
channel burned 2.74':
lidar invert = 2039.31
interpolated effective invert = 2036.57
END DESCRIPTION:
XS GIS Cut Line= 4
2206637.22852724410806.4412397822206207.61343548410702.982911562
2205774.49128175410717.0111594562205416.77096045410685.447601694
#Sta/Elev= 30
       0  2207.4    75.1 2159.31   103.9 2135.65   177.7 2078.51   198.6 2053.51
   223.3 2050.92   235.6 2043.57   243.8 2039.41   276.7 2039.06   317.9 2043.99
   333.5 2051.84   375.5 2052.76   400.2 2040.83   420.7 2041.24   445.3 2047.52
  480.55 2039.35   489.4 2036.57   536.1 2036.57   602.2 2036.57   687.2 2036.57
   709.4 2036.57   760.7 2036.58   805.5  2036.6   811.3 2039.76   833.5 2041.68
   856.8 2053.24   869.9 2056.09   905.7 2051.86  1094.9 2058.55  1234.4 2084.78
#Mann= 13 ,-1,0
       0      .1       0   103.9     .06       0   235.6     .04       0
   317.9     .06       0   400.2     .08       0  480.55    .035       0
   536.1    .016       0   602.2    .035       0   687.2    .016       0
   709.4    .035       0   760.7    .016       0   811.3     .08       0
   833.5     .05       0
#XS Ineff= 2 , 0
                          876.35          2068.4
Permanent Ineff=
       F       F
#Block Obstruct= 3 ,-1
   536.1   602.2 2049.94   687.2   709.4 2049.94   760.7     810 2049.94
Bank Sta=480.55,811.3
XS Rating Curve= 0 ,0
Exp/Cntr(USF)=0,0
Exp/Cntr=0.3,0.1

Type RM Length L Ch R = 1 ,60258   ,255.2,241.4,230
BEGIN DESCRIPTION:
channel burned 2.75' to transition to approximate zone:
lidar elevation = 2039.22
interpolated invert = 2036.47
END DESCRIPTION:
XS GIS Cut Line= 3
2206652.73332675410707.7429204732206311.16489226410645.342290903
2205400.01218832 410583.33105349
#Sta/Elev= 30
       0 2209.11    73.8 2161.12    98.2 2137.99   164.3 2084.18   191.5 2052.59
   195.7 2051.23   207.9 2051.54   216.1 2050.44   228.3 2042.52   248.6  2039.5
   289.3 2042.56   298.4  2042.7   313.7 2049.81   362.2 2052.84   394.3 2041.32
   418.4 2041.55   438.4 2046.19  495.37 2039.98   502.6 2036.47   787.2 2036.49
  801.94 2040.01   823.3 2044.98   843.4 2054.45   875.4 2056.72   890.7  2052.8
   900.9 2050.09  1055.8 2053.78  1099.9 2059.08  1179.8 2075.93  1260.5 2101.61
#Mann= 10 ,-1,0
       0      .1       0   195.7    .016       0   207.9      .1       0
   228.3     .04       0   289.3      .1       0  495.37    .035       0
  801.94      .1       0   890.7    .016       0   900.9     .05       0
  1099.9      .1       0
#XS Ineff= 2 , 0
                          868.39         2065.73
Permanent Ineff=
       F       F
Bank Sta=495.37,801.94
XS Rating Curve= 0 ,0
Exp/Cntr(USF)=0,0
Exp/Cntr=0.3,0.1

Type RM Length L Ch R = 1 ,60017   ,428.1,426.9,429.1
BEGIN DESCRIPTION:
channel burned 2.68' to transition to approximate zone:
lidar elevation = 2038.88
interpolated invert = 2036.20
END DESCRIPTION:
XS GIS Cut Line= 2
2206759.49415715410393.7975375912205430.32907518 410376.99269135
#Sta/Elev= 30
       0  2209.5    43.3 2181.16    71.3  2158.4   171.3 2094.65   199.3 2067.01
   223.3 2053.32   260.7 2049.48   276.5 2042.13   331.3 2039.26   339.3  2042.7
   351.5 2049.36   375.3 2041.22   398.9 2045.63   422.6 2041.97   535.4 2048.08
   571.4  2040.6   587.4 2045.46   610.5 2043.34   622.6 2040.23   631.4  2036.2
   859.4 2036.24   865.1 2040.17   911.4 2051.28   943.4 2056.45   979.4 2048.81
  1011.2 2051.13  1107.4 2051.46  1141.6 2056.44  1207.4  2077.9  1329.3 2133.24
#Mann= 10 ,-1,0
       0      .1       0   223.3     .06       0   276.5     .04       0
   339.3     .06       0   422.6      .1       0   610.5    .025       0
   622.6    .035       0   865.1      .1       0   911.4     .05       0
  1011.2      .1       0
Bank Sta=622.6,865.1
XS Rating Curve= 0 ,0
Exp/Cntr=0.3,0.1

Type RM Length L Ch R = 1 ,59590   ,492.9,510,523.6
BEGIN DESCRIPTION:
channel burned 1.98' to transition to approximate zone:
lidar elevation = 2037.69
interpolated invert = 2035.71
END DESCRIPTION:
XS GIS Cut Line= 3
2206806.19195252410057.9334369712206352.57299228409960.427887471
     2205580.699      409953.854
#Sta/Elev= 30
       0 2150.27    75.7  2111.6   120.7 2085.89   141.2 2064.61   153.4 2061.98
   165.7 2052.07   198.4 2048.99     213 2042.12     223 2038.82   308.9 2041.74
   349.8 2045.48   396.3 2043.92   419.9 2049.31     539 2049.65   552.4 2048.23
   568.4 2039.32   576.4 2039.53   592.4 2042.49  660.49    2038   664.4 2035.71
  877.04 2037.98   940.4 2055.65   964.4 2051.92   980.4 2053.63  1012.4 2069.07
  1064.4 2105.22  1128.4 2153.79  1144.4 2173.63  1205.3 2212.69  1235.9  2222.5
#Mann= 9 ,-1,0
       0      .1       0    75.7     .06       0     213     .04       0
   308.9      .1       0   576.4    .025       0  660.49    .035       0
  877.04      .1       0   964.4     .05       0  1064.4      .1       0
#XS Ineff= 2 , 0
       0                   948.8       0    2065
Permanent Ineff=
       F       F
Bank Sta=660.49,877.04
XS Rating Curve= 0 ,0
Exp/Cntr=0.3,0.1
