HEC-RAS study GRNBRRRV.prj: GRNBRRRV

--- GRNBRRRV.g01 (geometry) --- (continued)

Type RM Length L Ch R = 1 ,59080   ,485.3,481.9,482.2
BEGIN DESCRIPTION:
channel burned 1.59' to transition to approximate zone:
lidar elevation = 2036.72
interpolated invert = 2035.13
END DESCRIPTION:
XS GIS Cut Line= 3
2206877.53567802409499.1850152022206530.19204598409495.436445972
2205631.41097441409406.216678609
#Sta/Elev= 30
       0 2174.67    58.7 2128.25   141.4 2070.93   165.4 2049.91   193.4 2048.22
   201.4 2043.71   209.4 2037.96   253.4 2036.12   293.4 2042.64   309.4 2046.24
   341.4 2045.12   405.7 2044.18   446.3 2047.77     567 2050.99   622.7 2041.97
  711.79 2037.66   739.3 2035.13   904.1 2035.32  911.22 2037.49   928.2 2047.75
   940.3 2055.22   960.4 2059.15   972.4 2071.52   996.6 2090.49  1008.6 2106.07
  1020.4 2116.28    1085 2165.71  1119.1 2186.96  1173.4 2208.46  1250.6 2216.94
#Mann= 9 ,-1,0
       0      .1       0   141.4     .06       0   201.4     .04       0
   293.4      .1       0   341.4     .05       0   446.3      .1       0
  711.79    .035       0  911.22     .05       0   928.2      .1       0
Bank Sta=711.79,911.22
XS Rating Curve= 0 ,0
Exp/Cntr=0.3,0.1

Type RM Length L Ch R = 1 ,58598   ,565.1,504.4,459.2
BEGIN DESCRIPTION:
channel burned 1.96' to transition to approximate zone:
lidar elevation = 2036.53
interpolated invert = 2034.57
END DESCRIPTION:
XS GIS Cut Line= 4
2206763.32725891408879.2890497442206379.07509516 408996.71505535
2205974.31570567408955.7572599842205826.02259186 409001.08530865
#Sta/Elev= 30
       0 2140.76      32 2124.03    53.5 2114.07   132.2 2053.24   141.3 2049.44
     179 2047.59   191.5 2041.66   199.9 2036.78   254.3 2038.55   262.6 2041.75
     271 2045.62   324.4 2043.08   340.4 2043.54   416.8  2047.2   557.4 2048.52
   561.5 2047.82  573.05    2038   577.6 2034.74   742.4 2034.57   750.5 2034.57
  757.28 2037.87   778.6 2053.18   802.7 2055.79   806.8 2060.51   823.4 2087.94
   840.1  2105.5   865.2 2123.76   886.1 2134.32   907.6 2140.09   963.7 2148.44
#Mann= 10 ,-1,0
       0      .1       0      32     .06       0   132.2      .1       0
   191.5     .04       0   262.6      .1       0   324.4     .05       0
   340.4      .1       0  573.05    .035       0  757.28    .025       0
   840.1      .1       0
Bank Sta=573.05,757.28
XS Rating Curve= 0 ,0
Exp/Cntr=0.3,0.1

Type RM Length L Ch R = 1 ,58094   ,366.8,301.8,265.7
BEGIN DESCRIPTION:
channel burned 2.09' to transition to approximate zone:
lidar elevation = 2036.09
interpolated invert = 2034.0
END DESCRIPTION:
XS GIS Cut Line= 3
     2206465.082408255.2828971172206232.10888826408406.440945675
     2205619.802      408623.283
#Sta/Elev= 30
       0 2124.28    33.8  2102.8    59.9 2086.41    77.2 2066.96    96.4 2050.66
   125.1 2047.87   140.8  2041.3   143.7 2039.28   149.5 2036.58   175.5 2036.41
   206.1  2036.8   210.9 2039.46   218.9 2044.49   262.3 2046.66   294.6 2050.05
   311.6 2049.14   332.8  2042.7  341.09 2036.05   345.5  2034.1   519.5    2034
     545 2034.11   549.1 2036.03   578.9 2043.59   597.5 2045.88   615.1 2054.03
   634.1 2055.04   651.1 2069.95   680.5 2082.53   741.2 2097.44   927.3 2120.96
#Mann= 10 ,-1,0
       0      .1       0    33.8     .06       0   140.8      .1       0
   143.7     .04       0   210.9      .1       0   262.3    .025       0
  341.09    .035       0   549.1      .1       0   578.9    .025       0
   680.5      .1       0
Bank Sta=341.09,549.1
XS Rating Curve= 0 ,0
Exp/Cntr=0.3,0.1

Type RM Length L Ch R = 1 ,57792   ,303.3,269,262.7
BEGIN DESCRIPTION:
channel burned 2.16' to transition to approximate zone:
lidar elevation = 2035.81
interpolated invert = 2033.65
END DESCRIPTION:
XS GIS Cut Line= 4
2206526.34124837407970.1177197132206232.55892765407927.561496121
2206061.04986056408061.9136081922205632.19765027408454.626587281
#Sta/Elev= 30
       0 2213.96    55.7 2192.09      83 2177.71   165.1 2143.78   204.3 2131.55
   220.4 2123.28   228.7 2122.08   268.9 2094.09     285 2077.82   296.8 2070.19
   317.7 2064.18   329.6 2056.93   343.1 2052.03   415.1 2048.35     512 2046.76
   537.3 2042.56   555.1 2040.78   578.8 2040.45  589.24 2036.05   596.5 2033.72
   792.3 2033.65   800.8 2036.56   823.4 2041.23   857.6 2042.66   895.6 2052.84
   936.7  2057.7   962.1 2065.54   996.1 2080.68  1024.4 2087.64  1096.2 2100.33
#Mann= 6 ,-1,0
       0     .06       0   537.3      .1       0   555.1    .025       0
  589.24    .035       0   800.8    .025       0   936.7      .1       0
Bank Sta=589.24,800.8
XS Rating Curve= 0 ,0
Exp/Cntr(USF)=0,0
Exp/Cntr=0.3,0.1

Type RM Length L Ch R = 1 ,57523   ,405.8,420.4,434.1
BEGIN DESCRIPTION:
channel burned 1.72' to transition to approximate zone:
lidar elevation = 2035.06
interpolated invert = 2033.34
END DESCRIPTION:
XS GIS Cut Line= 2
2206118.87263049407534.2808326052205415.36226304 408360.66458615
#Sta/Elev= 30
       0 2129.85    84.4 2097.18    97.6 2088.58   121.4 2086.63   137.3  2078.8
   150.9 2077.18   182.7  2060.4   207.8 2051.87   266.5 2050.44   284.9  2046.3
   418.2 2045.13   455.6  2040.1   473.1 2045.13   486.4 2045.22   508.1 2038.49
   560.1 2037.74  621.87 2034.15   702.5 2033.34  762.34 2034.49   770.1 2039.93
   784.3 2043.08   802.3 2052.46   818.7 2053.78   835.4 2065.44   860.1 2068.17
     895 2068.07   954.6 2062.52   985.3 2063.43    1010 2064.74  1085.3 2075.81
#Mann= 5 ,-1,0
       0      .1       0   560.1    .025       0  621.87    .035       0
  762.34    .025       0   860.1      .1       0
Bank Sta=621.87,762.34
XS Rating Curve= 0 ,0
Exp/Cntr(USF)=0,0
Exp/Cntr=0.3,0.1

Type RM Length L Ch R = 1 ,57102   ,582.4,535.7,487.9
BEGIN DESCRIPTION:
channel burned 0.61' to transition to approximate zone:
lidar elevation = 2033.47
interpolated invert = 2032.86
END DESCRIPTION:
XS GIS Cut Line= 3
2205768.51492369407285.2725364592205639.42549651407522.234422204
 2205054.7218208 408050.35428208
#Sta/Elev= 30
       0  2154.6    27.2  2140.6   109.4 2110.41     173 2080.26   236.8 2042.63
   245.9 2043.25     255 2048.52   262.6 2049.91   313.9 2048.09   338.9 2044.53
   387.4 2044.81   414.4 2044.77   459.2 2035.15     498 2037.36   520.6 2034.71
   542.8 2032.86     686  2032.9   694.6 2034.52   707.5 2035.83     733  2042.9
   780.9 2042.64   837.8 2037.41   847.1 2040.32     865 2051.83   888.9 2053.07
   900.8 2058.38   924.7 2065.16   974.9  2074.1  1008.3  2076.2  1057.7 2082.69
#Mann= 5 ,-1,0
       0      .1       0   387.4    .025       0   520.6    .035       0
   694.6    .025       0   780.9      .1       0
Bank Sta=520.6,694.6
XS Rating Curve= 0 ,0
Exp/Cntr=0.3,0.1

Type RM Length L Ch R = 1 ,56567   ,494.9,480.7,467
XS GIS Cut Line= 2
2205137.00251102407088.4375652922204799.47584624407900.886078577
#Sta/Elev= 30
       0 2193.95    22.5 2187.37    43.9 2177.19    96.1 2135.24   104.8 2126.43
   117.8 2108.86   152.4 2052.91   156.7  2050.8   181.7 2050.14   187.9  2047.8
  207.03 2033.75     213 2032.25     382 2033.33   440.1 2036.96   463.3 2036.24
   512.2 2044.95   607.2 2040.78   637.5 2042.33   646.2 2041.15   656.1 2035.93
   671.4 2033.45   698.2    2034     702 2035.97   719.8 2042.55   758.8 2040.67
   789.1 2043.14   810.8  2051.9   828.1  2052.5   845.4 2061.08   879.8 2066.76
#Mann= 7 ,-1,0
       0      .1       0   181.7    .025       0  207.03    .035       0
     382    .025       0   440.1      .1       0   656.1     .04       0
     702      .1       0
Bank Sta=207.03,382
XS Rating Curve= 0 ,0
Exp/Cntr=0.3,0.1

Type RM Length L Ch R = 1 ,56086   ,487.9,494.1,502.9
XS GIS Cut Line= 2
2204628.61225551406979.6349768262204396.34107631407857.596540986
#Sta/Elev= 30
       0 2139.37    30.6 2133.93    55.4 2122.67    60.5 2117.76     105 2063.12
   117.5 2050.09   121.6 2047.23     134 2047.28   148.9 2045.03   161.72033.391
   167.1 2031.79   309.2 2031.89   316.6  2033.3   324.3 2038.36   332.6 2039.65
   365.7 2042.96   410.6 2041.83   518.8 2043.97   560.2 2043.22   576.7 2035.68
   593.3 2033.29   634.7 2033.45   639.7 2035.55   651.2 2039.73   692.6 2040.08
   717.4  2050.8   780.4 2054.93   855.6 2071.95   899.5 2083.86   908.2  2087.9
#Mann= 8 ,-1,0
       0     .12       0    30.6      .1       0     134    .025       0
   161.7    .035       0   316.6    .025       0   332.6      .1       0
   576.7     .04       0   639.7      .1       0
Bank Sta=161.7,316.6
XS Rating Curve= 0 ,0
Exp/Cntr=0.3,0.1

Type RM Length L Ch R = 1 ,55592   ,443,449,455.4
XS GIS Cut Line= 3
2204309.16964161  406782.86461732204164.94486336406871.728260522
 2203931.2365896407517.549795365
#Sta/Elev= 30
       0 2127.16    57.8 2120.89    76.3 2116.66    99.8 2104.79   150.7 2067.88
   170.9 2051.48   196.5 2050.06   210.5 2041.73   230.5 2033.07   230.5 2033.06
   230.5 2033.04     239 2031.34   434.7 2031.42     442 2033.16     456 2039.01
   481.5 2043.17   549.5 2042.89   558.5    2040   564.7 2035.78   570.8 2033.47
   596.3 2033.55   620.9 2034.51   623.8 2036.11   630.4 2039.59   642.8 2040.57
   714.6 2041.83     741 2050.53   762.2 2051.07   777.1 2056.13   856.2 2068.77
#Mann= 7 ,-1,0
       0      .1       0   150.7     .12       0   210.5    .025       0
   230.5    .035       0     442      .1       0   564.7     .04       0
   623.8      .1       0
Bank Sta=230.5,442
XS Rating Curve= 0 ,0
Exp/Cntr=0.3,0.1

Type RM Length L Ch R = 1 ,55143   ,240.5,330,421.5
XS GIS Cut Line= 3
2204203.62951825406551.2224711112203781.81559858 406654.82449609
2203504.41928321407299.569334088
#Sta/Elev= 30
       0 2085.65    40.6 2070.57    61.2 2065.29    73.6 2058.23   118.9 2057.06
   168.3 2049.64   201.3  2047.2   221.9  2035.4   229.3 2034.03   245.9 2031.66
   275.4 2031.83   282.2 2033.94   312.5 2036.69   421.1 2035.04     431 2036.52
   495.2 2033.77   583.5 2033.43   592.7 2031.88     598 2030.94 773.2912031.932
   780.9 2036.96   805.8 2042.77   833.1 2041.63   876.7 2036.15   906.3 2040.55
   951.9 2042.12   994.6 2050.09  1024.8 2050.57  1072.7 2066.86  1136.2 2092.12
#Mann= 7 ,-1,0
       0      .1       0   229.3     .04       0   282.2      .1       0
     431    .025       0   495.2     .05       0   592.7    .035       0
 773.291      .1       0
#XS Ineff= 2 , 0
                          805.28         2061.11
Permanent Ineff=
       F       F
Bank Sta=592.7,773.291
XS Rating Curve= 0 ,0
Exp/Cntr=0.3,0.1

Type RM Length L Ch R = 1 ,54813   ,367.5,408.2,446.3
XS GIS Cut Line= 4
2204219.30913292406527.7254217722203974.26116855406460.223049273
2203305.41814025406711.0685459362202993.28064161406714.465694745
#Sta/Elev= 30
       0 2089.85      53 2068.43    65.5 2060.14    94.5 2060.74   177.5 2048.99
     269 2041.39   277.8 2033.91   286.3 2031.69   313.9 2031.47   370.8 2033.62
   414.5 2036.42   440.1 2032.99   455.4 2036.64   482.8 2038.53   572.5 2036.33
   623.8 2032.51   644.2 2035.61   666.5 2034.53   685.3 2034.16719.37422031.877
   897.2 2030.56908.8067  2032.1   935.7 2048.22   965.6 2052.17   989.8 2075.08
  1037.8 2098.81  1073.8  2122.5  1081.8 2124.24  1173.6 2200.06  1280.7 2273.55
#Mann= 7 ,-1,0
       0      .1       0   277.8     .04       0   370.8      .1       0
   666.5     .05       0   685.3    .025       0719.3742    .035       0
908.8067      .1       0
Bank Sta=719.3742,908.8067
XS Rating Curve= 0 ,0
Exp/Cntr=0.3,0.1

Type RM Length L Ch R = 1 ,54405   ,174.2,213.5,246.7
XS GIS Cut Line= 4
2204255.53722841406338.4672108552203998.19412966406218.654036033
 2203683.0884473406264.5891762862202967.53166945406247.724201724
#Sta/Elev= 30
       0  2063.5    25.8 2067.67    69.4 2065.08   131.7 2053.68   215.5 2047.35
   314.2  2045.3   378.9 2039.46   392.1 2033.64   404.3  2030.3     488  2032.4
   552.7 2037.87   572.9 2035.72   677.2 2040.25   701.2 2038.71   713.2 2034.16
823.07922031.149   945.3 2030.03953.27922031.037   969.3 2033.92   993.3 2048.07
  1005.3 2049.11  1017.3 2054.91  1057.3  2085.6  1093.5 2124.03  1140.1 2164.85
  1153.4 2173.56  1165.4 2190.73  1189.4  2212.5  1245.6 2260.24  1318.1 2312.38
#Mann= 6 ,-1,0
       0      .1       0   392.1     .04       0     488      .1       0
823.0792    .035       0953.2792    .025       0   993.3      .1       0
Bank Sta=823.0792,953.2792
XS Rating Curve= 0 ,0
Exp/Cntr(USF)=0,0
Exp/Cntr=0.3,0.1

Type RM Length L Ch R = 1 ,54191   ,299.2,333.7,378.1
XS GIS Cut Line= 3
2204210.99007956406192.3122929092203726.45517528 406177.45070745
2203064.77920224405888.146494131
#Sta/Elev= 30
       0    2065   114.5 2049.12   266.9 2044.18     307 2038.77     328 2033.18
     343 2030.35     403  2031.8     443 2031.47     479 2038.13     496 2035.94
   513.4 2038.89   575.3 2040.64   645.2 2038.92   670.6 2037.18   696.3 2031.91
   705.5 2029.78   858.3 2029.75   874.8 2032.02   884.5 2035.17   897.6 2046.37
   923.8  2050.3   945.6 2070.76     998 2101.27  1024.2 2125.05  1044.6 2165.45
  1050.4 2172.89  1063.5 2180.92  1072.2 2189.99  1103.3 2212.28  1206.9 2305.59
#Mann= 6 ,-1,0
       0      .1       0     328     .04       0     403      .1       0
   645.2    .025       0   696.3    .035       0   874.8      .1       0
Bank Sta=696.3,874.8
XS Rating Curve= 0 ,0
Exp/Cntr(USF)=0,0
Exp/Cntr=0.3,0.1

Type RM Length L Ch R = 1 ,53857   ,296.3,322,356.8
XS GIS Cut Line= 4
2204276.97065193406158.5518474152203960.05547061405860.651576975
2203690.67756649405846.3903938162203324.64053206405497.783694366
#Sta/Elev= 30
       0 2074.23    60.4  2064.6   204.2 2051.38     259 2043.72   422.5  2043.7
     539 2037.23     547 2035.93   552.3 2031.23     555 2028.81   631.1 2028.41
   639.8 2031.28   655.1 2038.85   706.5  2039.9   741.3 2035.19   749.8 2031.79
   758.7 2029.31   929.1 2029.31   938.5 2031.83     962 2046.24   981.8 2049.61
   989.9 2065.12   996.5 2073.89  1019.7 2094.97  1035.5 2113.97  1075.1 2152.79
  1106.7 2194.82  1148.7 2228.24  1164.7 2251.45  1191.1 2271.93  1210.2 2280.93
#Mann= 6 ,-1,0
       0      .1       0   552.3     .04       0   639.8      .1       0
   749.8    .035       0   938.5    .025       0  1035.5      .1       0
Bank Sta=749.8,938.5
XS Rating Curve= 0 ,0
Exp/Cntr(USF)=0,0
Exp/Cntr=0.3,0.1

Type RM Length L Ch R = 1 ,53535   ,421.8,443.9,471.9
XS GIS Cut Line= 3
 2204348.0628132 406087.354862322203969.92901817 405750.65538285
 2203655.5973861405237.444564161
#Sta/Elev= 30
       0 2076.58    15.9 2076.39    63.4 2067.98   112.3    2062   298.9 2042.94
   444.4 2043.38   480.3  2042.1   512.7 2039.13   546.5 2040.42   563.3 2038.67
   573.7 2036.27   592.5 2034.94603.52592029.888   610.5 2028.27   831.7 2028.47
     839 2029.81     862 2041.94   883.3 2045.71   892.7  2051.5   897.4  2055.4
   902.1 2062.05   916.1 2088.94   924.6 2099.19   958.3 2132.65   976.8 2149.33
  1013.9 2179.94  1032.3 2196.49  1058.5  2222.9  1080.3 2247.53  1108.1 2273.92
#Mann= 4 ,-1,0
       0      .1       0603.5259    .035       0     839    .025       0
  886.31      .1       0
Bank Sta=603.5259,839
XS Rating Curve= 0 ,0
Exp/Cntr=0.3,0.1

Type RM Length L Ch R = 1 ,53091   ,490.3,497.8,510.2
XS GIS Cut Line= 2
2204467.94648785405956.6551814612204139.64148785405059.746539855
#Sta/Elev= 30
       0 2071.28    20.7 2067.94    88.9 2062.09   110.2 2057.45   152.2  2055.4
   161.3 2053.43   177.1 2052.01   273.8 2048.96   395.6 2040.87   451.5 2040.17
   485.8 2041.12   493.6 2039.85   502.1  2036.2   548.2 2028.14   553.2 2027.11
   569.5 2026.97   753.4    2027   758.7 2028.47   785.6 2043.49   804.5 2045.95
   808.8 2048.11   817.3 2060.04   825.7 2077.04   838.6 2098.46   842.8  2101.9
   885.4 2148.37   894.3 2159.95   906.8  2178.6   925.5 2201.55   955.1 2225.71
#Mann= 4 ,-1,0
       0      .1       0   548.2    .035       0   758.7    .025       0
     880      .1       0
Bank Sta=548.2,758.7
XS Rating Curve= 0 ,0
Exp/Cntr=0.3,0.1

Type RM Length L Ch R = 1 ,52594   ,500.7,500.4,501
XS GIS Cut Line= 2
2204895.61264161405816.0370531392204657.43664161404971.489002264
#Sta/Elev= 30
       0  2072.2    48.7 2065.98   156.7 2058.96     232  2050.9   302.2 2045.44
   318.8 2043.37   372.9 2041.43   390.9 2038.87   414.4 2038.24     431 2036.48
   451.8 2037.91   468.4 2033.74   501.7  2030.7   517.3 2027.53   530.8 2025.75
   701.2 2025.75   705.3 2025.87   709.5 2027.81   742.7 2043.33   755.2 2044.95
   759.4  2048.6   763.5 2053.53     776 2064.75   796.1 2086.13   802.6 2095.02
     830    2136   838.5 2145.75   846.6  2157.3   860.9 2175.28   877.5 2193.31
#Mann= 5 ,-1,0
       0     .06       0      90      .1       0   517.3    .035       0
   709.5    .025       0     820      .1       0
Bank Sta=517.3,709.5
XS Rating Curve= 0 ,0
Exp/Cntr=0.3,0.1

Type RM Length L Ch R = 1 ,52093   ,513.5,503.1,494.5
XS GIS Cut Line= 2
2205363.72694912405644.2132577742205147.23448785404859.897258906
#Sta/Elev= 30
       0 2066.73    69.5 2057.46    86.7 2056.67   214.8 2045.12   272.9 2041.56
   330.6 2039.46   343.4 2039.78   363.1 2038.74   401.5 2039.26   418.1 2032.52
   446.3 2027.03   451.3 2025.71   459.6 2025.38   654.6 2025.31   667.1 2025.75
     672 2027.19   675.4 2028.24   683.7 2034.49     692 2042.02   696.1  2043.4
   712.7 2045.06   720.8 2050.82   725.2 2055.02   738.6 2071.13   755.8 2088.13
   762.5 2093.95   783.3 2109.42   795.1 2119.72   808.2 2132.12   813.6 2138.92
#Mann= 4 ,-1,0
       0      .1       0   446.3    .035       0     672    .025       0
     740      .1       0
Bank Sta=446.3,672
XS Rating Curve= 0 ,0
Exp/Cntr=0.3,0.1

Type RM Length L Ch R = 1 ,51590   ,472.7,423.4,367.8
XS GIS Cut Line= 3
2205956.50953985405475.9846936142205808.07524213 405269.55567712
2205583.14492369404639.080950256
#Sta/Elev= 30
       0 2085.22   126.6 2063.25   185.7 2055.43   228.7 2051.08   251.6 2046.65
   267.4 2047.17   305.6 2043.11   380.5 2038.56   428.8 2038.87   445.8 2040.03
   462.8 2034.83     484 2030.41   489.2 2028.35   496.7 2025.25   501.8 2025.03
   723.8 2024.91   733.4 2025.36   738.8 2027.75     760 2041.87     777 2044.47
   781.3 2047.48   789.8 2056.29   796.4 2065.23   802.5 2071.81   819.5 2084.79
   836.1 2099.91   857.7  2125.2   864.9 2132.39   904.4 2155.75   923.7 2165.29
#Mann= 4 ,-1,0
       0      .1       0   489.2    .035       0   738.8    .025       0
  824.26      .1       0
Bank Sta=489.2,738.8
XS Rating Curve= 0 ,0
Exp/Cntr=0.3,0.1

Type RM Length L Ch R = 1 ,51167   ,677.2,548.7,436.9
XS GIS Cut Line= 3
 2206416.7245896405163.9380531392205930.94862822404582.910284234
2205711.18351215404513.326514417
#Sta/Elev= 30
       0 2133.04   110.3 2095.82     160 2080.79   195.4 2071.63   260.8 2056.85
   314.7 2047.69   326.9 2044.13   360.1 2040.94   391.4 2040.79   402.7  2036.3
   420.7 2033.11     434 2025.91   441.6 2024.69   691.8 2024.59     697 2025.62
   707.5 2031.01   724.3 2035.73     735 2041.52   764.1 2043.98   767.3 2045.19
   773.7 2052.17   786.4 2070.88     798 2082.39   814.8 2097.41   829.3 2108.61
   840.6 2114.45   859.7 2120.49   902.9 2130.48   961.6 2139.51   987.9 2142.29
#Mann= 5 ,-1,0
       0      .1       0     430    .025       0     434    .035       0
     697    .025       0  837.35      .1       0
Bank Sta=434,697
XS Rating Curve= 0 ,0
Exp/Cntr=0.3,0.1

Type RM Length L Ch R = 1 ,50618   ,599.4,527.8,469.4
XS GIS Cut Line= 3
     2206733.912      404228.5192206017.68278311404274.522177955
2205760.88551215404361.534539855
#Sta/Elev= 30
       0 2259.04     118 2175.51   158.1 2144.13   186.1 2123.92   230.2  2094.1
   262.3 2070.87   270.3 2064.92   278.3 2056.43   284.7 2051.71   298.4 2043.37
   310.4 2039.14   318.4 2034.79   326.4 2032.96   338.4 2026.07   342.4 2024.25
   346.4 2024.19   510.8 2024.22   522.8 2025.92   530.8 2031.25   553.7 2036.31
     603  2039.2   663.1 2037.61   683.1 2035.93   687.2 2036.18   699.2 2041.13
   719.3 2040.72   757.3 2047.33   821.9 2064.04   878.7 2084.07   988.8 2108.91
#Mann= 5 ,-1,0
       0      .1       0     290    .025       0   338.4    .035       0
   522.8    .025       0     690      .1       0
Bank Sta=338.4,522.8
XS Rating Curve= 0 ,0
Exp/Cntr=0.3,0.1

Type RM Length L Ch R = 1 ,50090   ,541.1,497.9,451.4
XS GIS Cut Line= 2
 2206276.3511515403634.2114115332205713.36028208404059.183667044
#Sta/Elev= 30
       0 2152.37    10.2 2140.48    25.3 2128.14    35.3 2117.34    40.3 2113.17
    55.3 2096.09    75.4    2078    85.4  2065.2   105.1 2050.74   116.5 2038.57
     125 2031.48   130.5 2029.12   144.4 2026.28   150.6 2023.58   155.6 2023.41
   295.9 2023.44   327.8 2026.24     345 2030.87   366.1 2031.57   376.1 2029.84
   384.9 2029.88   413.5 2030.71   423.2 2032.39   431.2 2031.97   473.5 2038.21
     483 2041.61   516.3  2040.2   621.7 2049.03   671.8 2057.51   705.4 2066.08
#Mann= 4 ,-1,0
       0      .1       0      40    .025       0   144.4    .035       0
   327.8      .1       0
#XS Ineff= 2 , 0
                          488.56          2050.6
Permanent Ineff=
       F       F
Bank Sta=144.4,327.8
XS Rating Curve= 0 ,0
Exp/Cntr=0.3,0.1

Type RM Length L Ch R = 1 ,49592   ,536.9,489,438.6
XS GIS Cut Line= 2
     2205947.474      403032.6742205483.31620464403910.558462409
#Sta/Elev= 30
       0 2204.47    17.6 2194.59    54.9 2178.82      67 2171.74   149.9 2130.63
   204.1    2106   224.8 2092.49   244.9  2082.4   258.5 2072.11   272.3 2056.76
   289.5 2047.65   304.7 2037.79   321.8 2031.78   335.4 2028.39   381.7 2023.88
   390.5 2022.72   525.4 2022.73   534.5 2024.06   561.6 2028.28   645.1 2026.02
   656.9 2029.59   677.6 2030.47   691.7 2034.03   701.9 2035.18   801.4 2039.35
   824.1 2041.42   842.2 2041.05   878.4  2043.8   926.3 2050.44     993 2064.92
#Mann= 7 ,-1,0
       0      .1       0     260    .025       0   381.7    .035       0
   534.5    .025       0     600      .1       0     710     .05       0
     820      .1       0
#XS Ineff= 2 , 0
                          596.57         2049.39
Permanent Ineff=
       F       F
Bank Sta=381.7,534.5
XS Rating Curve= 0 ,0
Exp/Cntr=0.3,0.1

Type RM Length L Ch R = 1 ,49103   ,526.1,510.8,497.9
XS GIS Cut Line= 2
     2205287.177      402864.6972205239.43169248403883.395975694
#Sta/Elev= 30
       0  2295.9    33.9    2271    48.5 2262.21    56.9 2255.28    68.6 2243.01
    88.6 2231.17   112.6 2214.39   124.6 2203.31   136.6 2189.31   192.7 2141.59
   200.7 2133.23   224.7 2115.41   272.8 2073.91     304 2050.81   328.8 2034.03
   346.1 2024.14   348.9 2022.51   356.9 2022.03   537.1 2022.09   549.1 2023.88
   581.3 2024.17     600 2027.84   633.2 2031.04   649.2 2034.67   693.2 2034.99
   721.3 2036.96   857.4 2040.74   889.5 2044.64   938.4  2058.3  1019.8 2076.32
#Mann= 6 ,-1,0
       0      .1       0     300    .025       0   346.1    .035       0
   581.3      .1       0     600     .05       0     800      .1       0
Bank Sta=346.1,581.3
XS Rating Curve= 0 ,0
Exp/Cntr=0.3,0.1

Type RM Length L Ch R = 1 ,48593   ,508.8,496.6,486.7
XS GIS Cut Line= 2
     2204735.406      402858.4882204779.98928208403866.290565292
#Sta/Elev= 30
       0 2269.19    18.7 2253.77    31.3 2241.56    62.8 2219.94    81.6 2198.02
    90.8 2189.95   131.9 2164.06   138.8 2158.44   146.8 2150.05   174.9 2128.64
   198.4 2108.29   210.9 2100.71   234.9 2079.88   250.9 2068.04   262.9 2056.83
     279 2044.74   294.7 2029.56     299 2026.69   306.2 2023.96     311 2021.38
   563.2 2021.41   571.7 2023.66   595.3 2027.32   615.3 2027.23   647.3 2033.97
   850.7 2036.71   879.6 2040.06   891.6 2039.86   911.6 2046.01  1008.8 2081.98
#Mann= 7 ,-1,0
       0      .1       0   306.2    .035       0   571.7      .1       0
     700     .05       0     800     .06       0     850     .05       0
     900      .1       0
Bank Sta=306.2,571.7
XS Rating Curve= 0 ,0
Exp/Cntr=0.3,0.1

Type RM Length L Ch R = 1 ,48096   ,522.2,501.7,480.9
XS GIS Cut Line= 2
     2204207.785      402905.2872204331.33653872403951.714642738
#Sta/Elev= 30
       0 2166.02      12 2158.96    32.1 2151.75    52.3 2148.05    72.4 2147.98
    92.5 2142.06   108.6 2139.76   136.4 2129.97   198.4 2098.79   217.4 2087.96
   246.1 2067.84   281.8 2037.08   289.9 2030.91   297.9 2026.06     310 2022.01
     310    2022   319.1 2020.43   587.5 2020.38     596 2020.49   601.9 2022.07
   640.3 2033.83   696.7  2033.7   761.1 2035.17   886.5 2035.03   915.3 2035.67
   929.7 2039.07   950.4 2038.25   962.5 2040.56   986.7 2050.33  1053.7 2086.53
#Mann= 5 ,-1,0
       0      .1       0     310    .035       0   601.9      .1       0
     660     .05       0     960      .1       0
Bank Sta=310,601.9
XS Rating Curve= 0 ,0
Exp/Cntr=0.3,0.1

Type RM Length L Ch R = 1 ,47594   ,519,499.4,484.5
XS GIS Cut Line= 2
     2203661.767      403021.8652203917.91351329404054.842488979
#Sta/Elev= 30
       0 2201.23    37.7 2182.91    61.1 2173.95   123.6 2152.79   176.5 2129.23
   196.3 2111.95   201.2 2106.24     226 2090.91   239.2 2081.63   275.5  2052.7
   283.7 2045.64   300.1 2027.53   308.5 2021.19   316.6 2018.73   324.6 2018.59
   584.5 2018.62   588.6 2019.26   591.7 2021.07     601 2025.92   617.5  2028.2
   628.9 2032.36   633.9 2033.01   877.1 2034.86   905.9 2036.04   918.3 2038.72
     943  2038.4   951.3  2040.1   967.8 2046.39  1021.3 2072.89  1064.3 2092.88
#Mann= 5 ,-1,0
       0      .1       0   308.5    .035       0   591.7      .1       0
     760     .05       0     940      .1       0
Bank Sta=308.5,591.7
XS Rating Curve= 0 ,0
Exp/Cntr=0.3,0.1

Type RM Length L Ch R = 1 ,47095   ,529.1,502.9,486
XS GIS Cut Line= 2
     2203139.469      403202.0982203484.99410288404116.986334088
#Sta/Elev= 30
       0 2295.05    33.2 2267.63   101.6 2218.91   137.9 2188.26   167.4 2159.39
   182.9 2145.81   187.2  2140.8     200 2118.33   204.3 2112.25   254.3  2058.4
   264.1 2049.19   285.4 2033.57   298.3 2019.78   302.6 2016.85   307.1 2016.56
   383.8 2016.53   520.7 2016.56   539.9 2019.94   559.1 2024.45   580.5 2026.72
   597.6 2032.03   614.7 2033.76     695 2031.66   730.2 2032.79   845.6 2032.66
   862.6 2037.93   888.4 2037.46   896.8 2039.57   965.3 2067.17     978 2071.25
#Mann= 5 ,-1,0
       0      .1       0   298.3    .035       0   539.9      .1       0
     590     .05       0     800      .1       0
Bank Sta=298.3,539.9
XS Rating Curve= 0 ,0
Exp/Cntr=0.3,0.1

Type RM Length L Ch R = 1 ,46592   ,517.5,505.9,497.4
XS GIS Cut Line= 2
      2202620.14      403444.9132203119.30435953404320.659154891
#Sta/Elev= 30
       0 2304.19    23.3 2284.15    64.8 2252.48      74 2237.75    78.6    2233
   110.8 2208.87   156.8 2176.91   207.5 2135.81   230.5 2110.69   239.7 2098.79
   246.6 2091.73   262.7 2068.65   299.6 2039.17     318 2022.11   325.7 2018.24
   340.4  2015.5   534.4 2015.51   543.6 2017.72   560.3 2024.03     575 2024.73
   594.2 2031.39   612.7 2032.82   694.7 2030.25   727.8 2031.41   800.8 2031.16
   847.5 2033.66   861.3 2037.34   877.1 2038.12   938.7 2057.09    1008 2080.83
#Mann= 5 ,-1,0
       0      .1       0   325.7    .035       0   543.6      .1       0
     590     .05       0     930      .1       0
Bank Sta=325.7,543.6
XS Rating Curve= 0 ,0
Exp/Cntr=0.3,0.1

Type RM Length L Ch R = 1 ,46086   ,480.4,493,505.9
XS GIS Cut Line= 2
     2202162.858      403735.744 2202723.9862312 404558.54530865
#Sta/Elev= 30
       0 2213.21    23.6 2196.61    50.9 2174.89    65.3 2167.78    88.3 2151.92
   125.8 2129.15   214.8 2077.45   229.4 2066.53   248.7 2055.45   272.1 2039.54
   282.6 2035.98   307.6 2024.22     333 2016.32   341.6 2014.82   479.8 2014.79
   528.8 2014.84   533.3 2016.51   543.1 2021.58   563.2 2023.31   577.9 2030.24
   584.5 2031.67   655.4 2029.09   769.1 2030.61     820  2033.1   834.5 2036.51
   853.9 2036.23   878.1 2042.96   923.1 2048.29   963.4 2055.23   995.9 2062.58
#Mann= 6 ,-1,0
       0      .1       0     333    .035       0   533.3      .1       0
     740     .05       0     860      .1       0     980     .05       0
Bank Sta=333,533.3
XS Rating Curve= 0 ,0
Exp/Cntr=0.3,0.1

Type RM Length L Ch R = 1 ,45593   ,474.1,495.5,511.5
XS GIS Cut Line= 2
     2201785.745      403992.8182202264.83110288404830.476641606
#Sta/Elev= 30
       0 2205.76      13 2203.94    40.2 2207.87    78.3 2208.94    95.9 2205.73
   107.6 2199.62   136.9 2175.95   139.8 2171.25   148.6  2148.5   151.5 2143.03
     166 2129.11   195.5 2103.81   206.3 2096.33   230.8 2072.97   262.7 2047.28
   309.8 2015.66   318.6 2014.09   391.6 2015.75   410.5 2014.27   567.8 2014.25
   576.4 2016.03   590.2 2025.31   605.9 2029.03     732 2030.05   774.6 2032.53
   793.5 2036.01     816 2035.79   842.8 2042.29   862.1 2044.04     965 2064.32
#Mann= 4 ,-1,0
       0      .1       0   309.8    .035       0   576.4     .05       0
     860      .1       0
#XS Ineff= 2 , 0
                          720.56         2047.42
Permanent Ineff=
       F       F
Bank Sta=309.8,576.4
XS Rating Curve= 0 ,0
Exp/Cntr=0.3,0.1

Type RM Length L Ch R = 1 ,45098   ,371.2,387.2,400.6
XS GIS Cut Line= 2
     2201396.576      404200.0562201778.15810288405100.601334088
#Sta/Elev= 30
       0  2207.7    22.9 2193.57    82.9  2146.6   101.1 2134.67   122.9  2115.6
   131.8 2106.89   142.5  2094.1   157.6 2082.66   170.6 2068.72   209.7 2039.48
   227.1 2031.43   244.5 2032.18   253.2 2030.57   274.3  2021.5   283.92016.026
   287.9 2013.88   292.3 2013.78   560.7 2013.84     566 2014.33   568.3 2016.03
   583.3 2026.09   600.7 2031.73   747.4 2030.64   783.2 2032.05     800 2035.16
   817.9  2035.5     831 2033.72   851.9  2040.6   870.1 2041.87   978.1 2060.41
#Mann= 6 ,-1,0
       0      .1       0     270    .025       0   283.9    .035       0
   568.3    .025       0     590     .05       0     800      .1       0
#XS Ineff= 2 , 0
                          811.83         2049.31
Permanent Ineff=
       F       F
Bank Sta=283.9,568.3
XS Rating Curve= 0 ,0
Exp/Cntr=0.3,0.1

Type RM Length L Ch R = 1 ,44710   ,671.6,698.1,730.6
XS GIS Cut Line= 2
2201071.90381498404300.5095906352201406.61477108405391.958360516
#Sta/Elev= 30
       0  2128.3    63.5 2088.19    97.2 2068.55   125.6 2048.54   151.3 2032.03
   172.2 2027.59   209.9 2023.99   260.1 2022.62   289.4 2016.95   301.9 2015.92
     327  2016.6   335.4 2014.77   343.8 2013.53     553 2013.56   561.3 2014.87
   573.9 2024.06   582.3  2025.9   590.6 2030.94     599 2033.37   737.1 2030.62
   759.6 2030.76     779 2033.06   799.8 2030.54   808.2 2028.22   820.7 2027.65
   887.7 2034.56   921.2 2042.56  1004.8 2073.07    1076 2094.14  1141.6 2116.34
#Mann= 4 ,-1,0
       0      .1       0   335.4    .035       0   561.3    .025       0
     570      .1       0
Bank Sta=335.4,561.3
XS Rating Curve= 0 ,0
Exp/Cntr(USF)=0,0
Exp/Cntr=0.3,0.1

Type RM Length L Ch R = 1 ,44012   ,430.9,420.9,418.9
XS GIS Cut Line= 3
2200577.11370597404159.833971406 2200494.6486878404339.316658009
2200581.96458939405615.098997914
#Sta/Elev= 30
       0 2152.79    59.7 2144.67    89.5 2135.02   111.5 2123.61   137.9 2103.56
   167.6 2084.73   207.4 2067.88   255.5 2043.19   279.5 2036.18   367.8 2022.79
   375.8  2016.4   379.8 2012.97   572.3    2013   611.1 2016.07   672.5 2017.67
   704.6 2020.53   720.6 2029.47   728.6 2030.93   813.3 2029.72   920.9 2031.22
   941.1 2033.38   965.2 2028.83   985.2  2030.5  1137.6 2027.47  1197.7    2033
  1213.8 2037.25  1257.9 2054.07    1318 2083.47  1377.2    2118  1476.3 2182.38
#Mann= 7 ,-1,0
       0      .1       0   375.8    .035       0   611.1      .1       0
  697.52     .05       0  897.52      .1       0  997.52     .05       0
 1197.52      .1       0
Bank Sta=375.8,611.1
XS Rating Curve= 0 ,0
Exp/Cntr(USF)=0,0
Exp/Cntr=0.3,0.1

Type RM Length L Ch R = 1 ,43591   ,509.4,497.8,488.4
XS GIS Cut Line= 2
     2200057.587      404245.8662200156.93869248405363.913823067
#Sta/Elev= 30
       0 2090.99    79.6 2056.42   123.8 2044.29   151.9 2040.06   220.2 2039.48
   256.3 2029.47   276.4 2026.39   308.5 2025.19   324.6 2015.44   328.6 2014.59
   380.8  2014.3   388.8 2012.69   545.5 2012.69   557.5 2014.62   569.5 2022.54
   585.6 2023.19   605.7  2029.3   649.9  2027.4   722.1  2029.5   794.4 2026.46
   814.5 2023.54   842.6 2031.53   854.7 2032.28   874.7 2024.69   890.8  2022.5
   902.9 2023.14     943 2032.16  1007.3 2056.62  1079.6  2080.7  1122.5 2097.63
#Mann= 4 ,-1,0
       0      .1       0   380.8    .035       0   557.5    .025       0
     600      .1       0
Bank Sta=380.8,557.5
XS Rating Curve= 0 ,0
Exp/Cntr=0.3,0.1

Type RM Length L Ch R = 1 ,43094   ,501.9,500.1,499.8
XS GIS Cut Line= 2
     2199527.545      404313.202     2199680.785      405210.207
#Sta/Elev= 30
       0 2062.74      56 2050.69    97.4 2037.92   117.7 2033.14     142 2031.34
   227.2 2030.36   275.9 2027.07   308.4 2028.44   312.5 2027.87   324.6 2020.29
   336.3 2015.22   340.8 2013.19     349 2012.41   539.7 2012.44   543.7 2012.69
   548.1 2015.38   555.9 2021.19   568.1 2026.61   572.1 2027.15   593.2 2026.22
     629 2027.24   718.2 2026.19   762.9 2026.87   787.2 2027.56   799.4 2029.28
   807.5 2032.17   819.7 2032.52   823.7 2033.36   860.3 2049.49     910 2075.92
#Mann= 4 ,-1,0
       0      .1       0   336.3    .035       0   548.1     .05       0
     740      .1       0
Bank Sta=336.3,548.1
XS Rating Curve= 0 ,0
Exp/Cntr=0.3,0.1

Type RM Length L Ch R = 1 ,42593   ,487,490.2,493.5
XS GIS Cut Line= 3
2198945.36064301403998.9764608682199040.40187856404445.581205657
     2199190.511      405293.965
#Sta/Elev= 30
       0 2063.84    47.2 2058.27    88.5 2049.68   109.6 2046.57   243.6 2035.21
   257.1 2032.71     274  2034.6   460.3 2029.88   667.4 2029.69   687.7 2028.46
   691.8 2027.31   708.1 2020.78   716.2 2014.97   720.2 2012.34   724.3 2012.12
   932.4 2012.17   935.5 2012.27   939.3 2015.49   947.7  2021.3   970.3 2024.91
  1024.9 2026.94  1085.8 2024.83  1134.6 2025.67  1138.6 2025.82  1150.8 2031.17
  1175.2 2031.86  1183.3 2036.41  1236.2 2072.76  1256.8 2088.47  1318.2  2139.3
#Mann= 4 ,-1,0
       0      .1       0  656.61     .05       0   716.2    .035       0
   939.3      .1       0
Bank Sta=716.2,939.3
XS Rating Curve= 0 ,0
Exp/Cntr=0.3,0.1

Type RM Length L Ch R = 1 ,42103   ,480.4,502.1,520.6
XS GIS Cut Line= 3
2198583.21697614403687.385808862  2198520.333551 404177.77503713
     2198698.196      405401.219
#Sta/Elev= 30
       0 2076.12    82.5 2061.66   102.6 2053.93   130.9 2046.01     143 2047.08
     272 2046.19   425.2 2039.95   788.9 2029.16     805 2027.25   841.4 2029.28
    1088 2028.72  1116.3 2024.01  1136.5 2015.471150.4862013.046  1156.7 2011.92
  1269.5 2011.88  1354.8 2011.941358.2782013.201  1366.9 2020.58  1379.5 2023.81
  1443.7 2023.52  1467.9 2026.67    1476 2030.31  1492.2 2031.65    1496 2033.63
  1520.7 2050.45  1543.9  2068.2  1577.1 2096.34  1633.7 2147.18  1730.7 2220.95
#Mann= 4 ,-1,0
       0      .1       01150.486    .035       01358.278    .025       0
  1364.4      .1       0
Bank Sta=1150.486,1358.278
XS Rating Curve= 0 ,0
Exp/Cntr=0.3,0.1

Type RM Length L Ch R = 1 ,41601   ,165.6,172.1,179.3
XS GIS Cut Line= 3
2198183.84457471403464.5360298662198132.10342992404232.057926051
     2198137.147      405468.842
#Sta/Elev= 30
       0  2086.1   117.1 2066.38     145 2058.62   189.1 2039.57   217.1 2032.47
   428.5 2032.39   886.4 2028.71  1206.4    2029  1286.4 2025.78  1370.4 2029.33
  1390.4 2027.99  1398.4 2025.58  1410.4 2018.72  1415.8 2013.67  1418.4 2011.75
  1422.4 2011.62  1654.4 2011.62  1658.4 2011.781661.3672014.005  1670.4 2020.49
  1678.4  2022.3  1690.4 2029.29  1706.4 2030.73  1718.2 2039.35  1814.6 2120.75
  1878.4 2177.04  1930.4 2225.45  1982.4 2269.45  1995.3 2285.49  2006.1 2295.62
#Mann= 6 ,-1,0
       0      .1       0     390     .08       0  789.26      .1       0
  1415.8    .035       01661.367    .025       0 1669.26      .1       0
Bank Sta=1415.8,1661.367
XS Rating Curve= 0 ,0
Exp/Cntr=0.3,0.1

Type RM Length L Ch R = 1 ,41429   ,315.5,335.2,356
XS GIS Cut Line= 3
 2198131.2188518403420.2398845832198035.83439335403587.807176456
2197939.45644002405482.899032954
#Sta/Elev= 30
       0 2092.99   111.3 2077.53   161.3 2067.79   184.8 2060.01   230.2 2040.82
   253.7 2034.41   274.3  2031.1  1007.2 2027.97  1231.5 2028.99  1283.6 2028.35
  1351.7 2025.25  1427.8 2028.69  1463.8 2025.74  1483.9 2014.96  1504.9 2012.89
  1511.9 2011.53  1708.1 2011.53    17122012.874  1744.2 2029.43  1756.2 2029.81
  1760.3 2031.32    1825 2090.39  2024.5 2254.62  2028.6  2258.4  2040.6 2278.67
  2044.6 2283.27  2052.6 2287.15  2060.6  2294.1  2080.6 2317.21  2090.4 2322.23
#Mann= 6 ,-1,0
       0      .1       0  462.81     .08       0  852.81      .1       0
 1442.81    .025       0  1504.9    .035       0    1712      .1       0
Bank Sta=1504.9,1712
XS Rating Curve= 0 ,0
Exp/Cntr(USF)=0,0
Exp/Cntr=0.3,0.1

Type RM Length L Ch R = 1 ,41094   ,500.2,506.3,512.2
XS GIS Cut Line= 3
2197962.87201368403310.6316060232197774.50824831404301.832595635
     2197536.955      405381.501
#Sta/Elev= 30
       0 2088.25      27 2082.53      84  2075.3   177.7 2069.59   267.2 2059.28
   295.7 2051.97   332.4  2035.6   352.7 2033.09   450.5 2029.01  1122.9 2026.83
    1340 2029.03  1417.8 2024.25  1495.7 2026.68  1524.3 2025.31  1528.4 2023.49
 1535.26 2013.63  1540.7 2011.35  1749.6 2011.341757.683 2013.51  1765.7 2017.63
  1778.3 2020.61  1790.5 2028.61  1806.9  2029.8    1811 2032.49  1835.6  2055.8
  1916.8 2110.85  2073.1 2231.88  2093.6 2250.43  2101.8 2262.75  2114.4 2275.44
#Mann= 8 ,-1,0
       0      .1       0     460     .08       0     660      .1       0
     760     .08       0     860      .1       0 1458.94    .025       0
 1535.26    .035       01757.683      .1       0
Bank Sta=1535.26,1757.683
XS Rating Curve= 0 ,0
Exp/Cntr=0.3,0.1

Type RM Length L Ch R = 1 ,40588   ,504.2,506.7,511.9
XS GIS Cut Line= 2
2197509.86454806403458.220333944     2197027.295      405245.093
#Sta/Elev= 30
       0 2081.84    40.4 2076.81    78.8 2067.63   101.7 2058.07   131.5 2041.13
   152.2 2033.61   181.2  2028.6   206.1 2026.56   359.3  2025.5     840 2026.89
    1130 2028.01    1188 2022.94  1246.1 2025.24  1270.9  2023.41299.5382013.224
  1308.2  2011.1  1511.2 2011.061515.1372012.897  1519.5 2017.22  1531.9 2019.04
  1548.5  2027.4  1569.2 2030.11  1594.1 2046.64  1657.8 2094.21    1706 2131.55
  1736.1 2157.68  1786.1 2206.95  1811.1 2228.98  1824.1  2247.7  1850.9 2271.16
#Mann= 10 ,-1,0
       0      .1       0     310     .08       0     410      .1       0
     620     .05       0     820      .1       0     840     .05       0
    1130      .1       0    1230    .025       01299.538    .035       0
1515.137      .1       0
Bank Sta=1299.538,1515.137
XS Rating Curve= 0 ,0
Exp/Cntr=0.3,0.1

Type RM Length L Ch R = 1 ,40081   ,496.5,491.2,488.2
XS GIS Cut Line= 2
2197052.94358987403399.700849416     2196529.747      405081.422
#Sta/Elev= 30
       0  2056.4    72.1 2048.78   127.2    2032   174.3 2029.17   407.9 2022.83
   424.6 2025.41   596.4 2023.72   688.6 2025.81   893.8 2025.02  1048.8 2027.04
  1157.7 2025.27  1161.9 2023.57  1170.3 2014.541175.0582012.343  1199.6 2010.67
  1249.9 2013.99  1279.2 2010.721444.8052012.106  1463.5 2019.41  1476.1 2020.65
  1487.5 2025.74  1505.4 2028.57  1530.6 2028.39    1561 2049.89    1576 2058.39
    1606  2066.9  1666.4 2054.01  1714.9 2051.64  1743.1 2044.32  1761.2 2042.57
#Mann= 5 ,-1,0
       0      .1       0     380     .05       0    1100      .1       0
1175.058    .035       01444.805      .1       0
Bank Sta=1175.058,1444.805
XS Rating Curve= 0 ,0
Exp/Cntr=0.3,0.1

Type RM Length L Ch R = 1 ,39590   ,539.5,516.1,507.1
XS GIS Cut Line= 2
 2196569.8696931 403172.65724161     2196074.686      404933.269
#Sta/Elev= 30
       0 2082.87    33.8 2078.66    54.6 2073.68    83.6 2063.83   104.4 2053.41
   116.9 2051.88   129.4 2045.48   147.7 2039.98   237.4  2032.3   353.7 2027.95
   661.2 2024.44    1056 2026.31  1091.5 2023.44  1105.8 2017.61  1130.4 2018.17
    1164 2013.87  1172.3  2015.7  1188.8 2012.76  1222.2 2012.09  1234.6 2010.28
  1483.9 2010.31  1489.9 2012.03  1503.3 2016.75  1521.3 2019.29  1533.8 2024.87
  1571.2 2023.72  1603.9 2031.01  1674.9 2083.05  1762.3 2160.89  1828.9 2212.57
#Mann= 10 ,-1,0
       0      .1       0     200     .08       0     510     .05       0
     710     .08       0     970     .05       0    1020     .06       0
    1120      .1       0    1220    .025       0  1222.2    .035       0
  1489.9      .1       0
Bank Sta=1222.2,1489.9
XS Rating Curve= 0 ,0
Exp/Cntr=0.3,0.1

Type RM Length L Ch R = 1 ,39074   ,539.3,527.2,518.3
XS GIS Cut Line= 2
2195941.73387563402944.3607789892195626.87865229404792.399670774
#Sta/Elev= 30
       0 2099.73    21.1 2092.25    41.4 2082.56    77.9 2064.18   118.5 2041.02
   151.1 2027.27   163.1 2024.35   532.4 2022.56   759.6 2026.19     861 2023.82
  1009.6 2024.66  1092.3 2023.21  1193.8 2026.76  1214.1 2025.66  1222.4 2020.05
  1234.4 2015.82 1240.61 2011.95  1246.5 2009.91  1502.2 2009.94  1509.7 2011.95
  1518.4 2015.01  1530.6 2015.43  1550.8 2025.16  1640.1 2021.16  1664.5 2023.28
  1680.7 2028.44    1705 2030.03  1749.7 2048.77  1782.1 2065.85  1874.7 2121.01
#Mann= 10 ,-1,0
       0      .1       0     330     .08       0     530      .1       0
     630     .08       0     750     .05       0    1030      .1       0
    1130    .025       0 1240.61    .035       0  1509.7    .025       0
    1520      .1       0
Bank Sta=1240.61,1509.7
XS Rating Curve= 0 ,0
Exp/Cntr=0.3,0.1

Type RM Length L Ch R = 1 ,38546   ,450.5,459.5,498
XS GIS Cut Line= 3
2195579.20147734402931.4871947912195218.99612667 403996.26867933
2195133.78965845404696.384316904
#Sta/Elev= 30
       0 2096.14    39.8 2069.82    73.6 2052.64     120  2034.2   141.1 2027.88
   166.5 2023.93   478.9 2020.29   609.9  2023.3   943.4 2025.82   985.7 2022.36
  1051.3 2021.62  1074.3 2018.09    1087 2019.95  1141.8 2010.77  1149.2  2009.5
  1188.5 2009.56  1209.6  2011.9  1245.9 2009.53  1511.8 2010.74  1511.8 2010.75
  1511.8 2010.77  1523.9 2015.28  1612.8 2020.87    1673 2020.87  1689.1 2015.47
  1701.2 2019.99  1725.4 2021.42  1737.5 2027.01  1753.6 2028.63  1829.3 2097.14
#Mann= 8 ,-1,0
       0      .1       0     460     .08       0     560     .05       0
     770     .08       0     870      .1       0  1141.8    .035       0
  1511.8    .025       0 1574.06      .1       0
Bank Sta=1141.8,1511.8
XS Rating Curve= 0 ,0
Exp/Cntr=0.3,0.1

Type RM Length L Ch R = 1 ,38087   ,459.9,457,453.1
XS GIS Cut Line= 5
2195276.28408971402942.8066924362194996.20960377403633.444913451
2194798.88439776403821.2221256172194788.01900682403864.944224304
2194626.15768026 404796.18407834
#Sta/Elev= 30
       0 2071.27    67.3 2034.82   140.7 2021.47   265.9 2019.97     404 2022.37
   563.2 2022.41   671.4 2022.72   750.8 2025.19   872.5 2018.99   892.2  2014.3
   903.5 2008.97   959.6 2008.84   965.4 2014.94   971.2 2021.24   982.7 2025.53
  1164.4 2025.691183.3232012.222  1188.8 2008.75  1477.8 2011.65  1536.6 2019.88
  1554.2 2019.58  1562.3 2014.12  1574.7 2008.721669.9132011.383  1751.2 2031.43
  1781.6 2052.62  1838.4 2101.85  1862.8 2138.25  1887.1 2160.82  2007.9 2219.89
#Mann= 12 ,-1,0
       0      .1       0   140.7     .08       0   265.9      .1       0
     404     .05       0   563.2     .08       0   671.4      .1       0
   892.2     .04       0   965.4      .1       01183.323    .035       0
  1477.8      .1       0  1562.3    .035       01669.913      .1       0
Bank Sta=1183.323,1669.913
XS Rating Curve= 0 ,0
Exp/Cntr=0.3,0.1

Type RM Length L Ch R = 1 ,37630   ,499,529.7,595.7
XS GIS Cut Line= 2
2194487.15740239402793.5513850072194224.55567694404497.355664613
#Sta/Elev= 30
       0 2127.02    96.8 2062.78   137.2  2043.5   181.7 2030.18   226.3    2020
   282.9 2019.15     550 2024.27   566.9  2011.9   574.3 2007.91     623 2008.08
     631  2011.7   699.8 2022.77   845.5 2023.18  1116.7 2020.27  1157.1 2009.92
  1310.9    2008  1345.3 2014.24  1412.1 2021.35  1432.3 2020.25  1440.1 2014.41
  1444.5 2009.69  1460.7 2008.04  1555.8 2009.92  1570.1 2015.71  1586.1 2024.83
  1618.9 2034.59  1642.8 2053.31  1679.2 2089.79  1691.4 2097.08  1723.9 2130.34
#Mann= 10 ,-1,0
       0      .1       0   181.7     .08       0   282.9      .1       0
   566.9     .04       0     631      .1       0  1157.1    .035       0
  1345.3      .1       0  1440.1    .035       0  1555.8    .025       0
  1570.1      .1       0
Bank Sta=1157.1,1555.8
XS Rating Curve= 0 ,0
Exp/Cntr=0.3,0.1

Type RM Length L Ch R = 1 ,37100   ,629.9,623.7,621.7
XS GIS Cut Line= 3
2194097.50679565402801.9209253172193881.62296554403688.175287618
     2193608.188      404373.224
#Sta/Elev= 30
       0 2113.07   126.3 2033.72   174.6 2021.86     201 2017.89   233.9 2021.28
   386.2  2021.6   435.6  2011.5   480.9 2007.56   489.2 2011.97   571.5 2021.94
   740.3 2021.79   789.7 2012.49   843.2  2017.9  1012.3 2018.89  1033.8 2012.56
  1068.3  2015.3  1081.2 2009.47  1292.7 2007.51  1305.2 2009.62  1360.4 2028.44
  1378.4 2044.63  1412.4 2048.89  1437.4 2060.82  1486.1 2094.51  1606.7 2191.35
  1615.3 2223.03  1619.6 2231.87  1640.5 2241.26  1645.4 2251.56  1649.8 2252.92
#Mann= 9 ,-1,0
       0      .1       0   174.6     .08       0   233.9      .1       0
   435.6     .04       0   489.2      .1       0  1012.3    .025       0
  1081.2    .035       0  1305.2    .025       0  1412.4      .1       0
Bank Sta=1081.2,1305.2
XS Rating Curve= 0 ,0
Exp/Cntr=0.3,0.1

Type RM Length L Ch R = 1 ,36477   ,373.8,381,385.8
XS GIS Cut Line= 2
2193556.47043697402727.1697365672193070.46471679404080.028563029
#Sta/Elev= 30
       0 2138.64    39.3 2104.73   112.6 2050.54   155.1 2023.64   176.4  2017.3
   273.8 2017.43   312.4 2020.41   439.6  2023.2   652.2 2023.03   745.9 2019.46
   809.7 2012.98   843.7 2013.55   864.9 2009.49   886.2 2010.63   898.9 2008.87
   911.6 2006.91  1115.7 2008.12  1132.7 2009.87  1162.5  2024.5  1183.8 2025.23
  1196.3 2031.99    1222 2050.41  1345.2 2149.89    1362 2166.93  1387.7 2186.56
    1392 2191.93  1396.2 2212.82  1400.5  2222.2  1415.2 2238.46  1437.5 2251.06
#Mann= 4 ,-1,0
       0      .1       0     890    .025       0   898.9    .035       0
  1115.7      .1       0
Bank Sta=898.9,1115.7
XS Rating Curve= 0 ,0
Exp/Cntr=0.3,0.1

Type RM Length L Ch R = 1 ,36095   ,433.8,503.2,551.8
XS GIS Cut Line= 2
2193209.12528434402693.446968903     2192676.463      403989.548
#Sta/Elev= 30
       0 2119.72    51.6 2075.93   112.2 2032.12   120.8  2023.9   133.8 2022.68
   151.1 2015.43   246.2 2015.94   306.8 2020.09   435.8 2022.55     730 2021.41
   757.6 2021.58   786.8 2012.72   795.4 2007.85   804.1 2006.62  1033.3 2007.76
  1050.6 2014.91  1064.1 2024.01  1079.4    2026  1085.2 2029.28  1116.2 2058.27
  1171.7 2104.59  1206.3 2131.16  1210.6 2136.64  1214.9 2144.95  1219.3 2150.99
  1232.2 2159.27  1254.7 2166.78  1288.4 2173.39  1328.4 2173.44  1401.3 2169.98
#Mann= 5 ,-1,0
       0      .1       0     730    .025       0   795.4    .035       0
  1033.3    .025       0    1040      .1       0
Bank Sta=795.4,1033.3
XS Rating Curve= 0 ,0
Exp/Cntr=0.3,0.1

Type RM Length L Ch R = 1 ,35592   ,465.7,499.2,527.1
XS GIS Cut Line= 4
2192921.57205314 402568.527174672192703.99000736403026.514060358
2192164.95796539403550.9625109512191882.38666655403854.855756229
#Sta/Elev= 30
       0  2131.7    67.6 2076.68   111.4 2044.07   139.6 2024.89   151.6 2023.14
     169 2015.43   315.1 2016.44   370.8 2020.44   707.7 2021.81   717.4 2019.51
   734.52009.548   746.4 2006.28   986.7 2006.31   989.7 2008.29    1018 2023.38
  1040.6  2026.5    1117 2099.84  1131.1 2119.53  1170.9 2162.38  1204.7 2183.98
  1222.1 2201.47  1266.1  2218.3  1377.7 2238.34  1407.1 2240.39  1524.3 2228.75
  1592.4 2211.97  1606.2 2206.19  1618.6 2205.48  1640.5 2216.88  1674.1 2226.38
#Mann= 4 ,-1,0
       0      .1       0  697.04    .025       0   734.5    .035       0
   989.7      .1       0
Bank Sta=734.5,989.7
XS Rating Curve= 0 ,0
Exp/Cntr=0.3,0.1

Type RM Length L Ch R = 1 ,35093   ,478.6,501.5,520.7
XS GIS Cut Line= 2
2192731.74110515402512.287921423     2191748.016      403135.703
#Sta/Elev= 30
       0 2092.56    32.2 2069.44    56.3 2054.89    98.9 2032.54   121.2 2023.22
   133.7 2023.02   174.2 2016.32   263.2 2015.48   278.9 2013.48   547.2 2020.18
     554 2018.95   571.4  2007.1   577.2 2005.34   823.6 2005.34   829.3 2006.57
   835.1 2010.61   847.2 2014.69   856.6 2022.75     876 2025.62   894.5 2041.94
   916.3 2055.36   945.3 2072.28   958.2 2076.79     975 2087.61  1017.9 2109.31
  1093.1 2143.27  1107.6 2144.31  1122.1 2151.55  1140.8 2156.87  1164.6 2166.78
#Mann= 5 ,-1,0
       0      .1       0     550    .025       0   571.4    .035       0
   829.3     .05       0     900      .1       0
Bank Sta=571.4,829.3
XS Rating Curve= 0 ,0
Exp/Cntr=0.3,0.1

Type RM Length L Ch R = 1 ,34591   ,480,497.7,514.7
XS GIS Cut Line= 2
2192508.33600226402174.401563029     2191488.849      402633.143
#Sta/Elev= 30
       0 2131.01    70.4 2092.52   171.2 2040.93   210.7 2023.57   223.9 2022.21
     237 2018.69   254.6 2018.62   263.4 2016.92   276.5 2018.52     430 2014.77
   478.3 2017.15   495.8 2011.24   510.4  2011.8   522.1 2005.38   530.9 2004.31
   767.1 2005.24   789.7 2011.09   806.9 2012.08   824.8 2015.92   842.3 2023.14
   864.3 2024.34   868.7 2026.32   912.8 2053.82   960.8 2088.27   973.9 2099.05
   997.5 2113.85    1009 2123.77    1088 2182.71  1109.9 2201.59  1117.9 2206.81
#Mann= 6 ,-1,0
       0      .1       0     480    .025       0   522.1    .035       0
   767.1    .025       0     800     .05       0     910      .1       0
Bank Sta=522.1,767.1
XS Rating Curve= 0 ,0
Exp/Cntr=0.3,0.1
